--- EIGHTEENMILE CREEK.prj (project) ---

Proj Title=EIGHTEENMILE CREEK Base Level Engineering
Current Plan=p01
Default Exp/Contr=0.3,0.1
English Units
Geom File=g01
Flow File=f01
Plan File=p01
Y Axis Title=Elevation
X Axis Title(PF)=Main Channel Distance
X Axis Title(XS)=Station
BEGIN DESCRIPTION:
EIGHTEENMILE CREEK
END DESCRIPTION:
DSS Export Rating Curves= 0
DSS Export Rating Curve Sorted= 0
DSS Export Volume Flow Curves= 0
DXF OffsetX= 0
DXF OffsetY= 0
DXF ScaleX= 1
DXF ScaleY= 10

--- EIGHTEENMILE CREEK.p01 (plan) ---

Plan Title=Multiple Run
Short Identifier=Multiple
Geom File=g01
Flow File=f01
Subcritical Flow
K Sum by GR= 0
Std Step Tol= 0.01
Critical Tol= 0.01
Num of Std Step Trials= 20
Max Error Tol= 0.3
Flow Tol Ratio= 0.001
Split Flow NTrial= 30
Split Flow Tol= 0.02
Split Flow Ratio= 0.02
Log Output Level= 0
Friction Slope Method= 1
Unsteady Friction Slope Method= 2
Unsteady Bridges Friction Slope Method= 1
Parabolic Critical Depth
Global Vel Dist=  1 , 1 , 1
Global Log Level= 0
CheckData=True
Encroach Param= -1, 0, 0, 0
BEGIN DESCRIPTION:
Multiple Run
END DESCRIPTION:

--- EIGHTEENMILE CREEK.f01 (steady flow) ---

Flow Title=Multiple
Program Version=4.10
Number of Profiles= 7
Profile Names=10-year,25-year,50-year,1pct_min,100-year,1pct_plu,500-year
River Rch & RM=EIGHTEENMILE CRE,Reach-1         ,87005
    1149    1914    2625    1739    3471    6925    6008
River Rch & RM=EIGHTEENMILE CRE,Reach-1         ,83163
    1260    2106    2893    1919    3830    7641    6647
River Rch & RM=EIGHTEENMILE CRE,Reach-1         ,79743
    1564    2641    3656    2441    4871    9718    8568
River Rch & RM=EIGHTEENMILE CRE,Reach-1         ,78691
    1674    2828    3915    2613    5214   10403    9167
River Rch & RM=EIGHTEENMILE CRE,Reach-1         ,74501
    1776    3005    4164    2782    5551   11076    9776
River Rch & RM=EIGHTEENMILE CRE,Reach-1         ,70701
    2544    4373    6125    4131    8243   16447   14798
River Rch & RM=EIGHTEENMILE CRE,Reach-1         ,68646
    2629    4521    6333    4271    8523   17005   15298
River Rch & RM=EIGHTEENMILE CRE,Reach-1         ,65576
    2732    4701    6588    4444    8867   17693   15923
River Rch & RM=EIGHTEENMILE CRE,Reach-1         ,62710
    3701    6438    9089    6172   12316   24573   22412
River Rch & RM=EIGHTEENMILE CRE,Reach-1         ,59137
    4104    7153   10111    6873   13713   27361   24998
River Rch & RM=EIGHTEENMILE CRE,Reach-1         ,55036
    4188    7299   10316    7011   13988   27911   25490
River Rch & RM=EIGHTEENMILE CRE,Reach-1         ,51153
    4572    7980   11292    7680   15324   30575   27965
River Rch & RM=EIGHTEENMILE CRE,Reach-1         ,47187
    4649    8114   11481    7808   15579   31084   28424
River Rch & RM=EIGHTEENMILE CRE,Reach-1         ,43428
    5771   10108   14342    9776   19506   38920   35737
River Rch & RM=EIGHTEENMILE CRE,Reach-1         ,40630
    6467   11363   16156   11033   22015   43925   40480
River Rch & RM=EIGHTEENMILE CRE,Reach-1         ,38610
    6460   11338   16110   10994   21936   43768   40276
River Rch & RM=EIGHTEENMILE CRE,Reach-1         ,34994
    6466   11332   16084   10964   21876   43649   40075
River Rch & RM=EIGHTEENMILE CRE,Reach-1         ,30840
    6765   11872   16865   11506   22957   45806   42120
River Rch & RM=EIGHTEENMILE CRE,Reach-1         ,29271
    7009   12305   17487   11933   23809   47506   43703
River Rch & RM=EIGHTEENMILE CRE,Reach-1         ,26853
    7199   12643   17971   12265   24472   48828   44932
River Rch & RM=EIGHTEENMILE CRE,Reach-1         ,24290
    7225   12679   18013   12287   24516   48916   44964
River Rch & RM=EIGHTEENMILE CRE,Reach-1         ,21101
    7295   12797   18177   12395   24732   49346   45331
River Rch & RM=EIGHTEENMILE CRE,Reach-1         ,17891
    7346   12881   18290   12468   24877   49637   45566
River Rch & RM=EIGHTEENMILE CRE,Reach-1         ,14589
    7329   12848   18239   12431   24803   49488   45409
River Rch & RM=EIGHTEENMILE CRE,Reach-1         ,13208
    8135   14292   20320   13867   27668   55205   50781
River Rch & RM=EIGHTEENMILE CRE,Reach-1         ,9146
    8317   14615   20783   14185   28302   56470   51957
River Rch & RM=EIGHTEENMILE CRE,Reach-1         ,6393
    8804   15443   21938   14958   29844   59547   54649
River Rch & RM=EIGHTEENMILE CRE,Reach-1         ,3376
    8797   15420   21897   14923   29776   59410   54474
Boundary for River Rch & Prof#=EIGHTEENMILE CRE,Reach-1         , 1
Up Type= 0
Dn Type= 3
Dn Slope=0.00127
Boundary for River Rch & Prof#=EIGHTEENMILE CRE,Reach-1         , 2
Up Type= 0
Dn Type= 3
Dn Slope=0.00127
Boundary for River Rch & Prof#=EIGHTEENMILE CRE,Reach-1         , 3
Up Type= 0
Dn Type= 3
Dn Slope=0.00127
Boundary for River Rch & Prof#=EIGHTEENMILE CRE,Reach-1         , 4
Up Type= 0
Dn Type= 3
Dn Slope=0.00127
Boundary for River Rch & Prof#=EIGHTEENMILE CRE,Reach-1         , 5
Up Type= 0
Dn Type= 3
Dn Slope=0.00127
Boundary for River Rch & Prof#=EIGHTEENMILE CRE,Reach-1         , 6
Up Type= 0
Dn Type= 3
Dn Slope=0.00127
Boundary for River Rch & Prof#=EIGHTEENMILE CRE,Reach-1         , 7
Up Type= 0
Dn Type= 3
Dn Slope=0.00127
DSS Import GetInterval= 0
DSS Import GetPeak= 0
DSS Import FillOption= 0

--- EIGHTEENMILE CREEK.g01 (geometry) ---

Geom Title=Existing Conditions
Program Version=4.10

River Reach=EIGHTEENMILE CRE,Reach-1
Reach XY= 30
        2450425.       13508525.      2451085.47     13506764.46
      2453069.54     13505077.46      2453801.42     13502297.85
      2455740.18     13502875.43      2457485.47     13501725.93
      2459031.35     13502267.58       2460365.2     13500235.48
      2461964.53     13499984.82        2464725.       13494725.
      2467564.32     13494625.75      2468840.18     13495525.44
       2470709.8      13494675.5      2471371.66     13495567.01
      2473714.56     13495176.05      2474874.91     13496167.65
       2478359.6     13495425.09        2481575.     13496967.44
       2483878.3     13496083.08      2484626.28     13497171.63
      2486258.36     13497008.29      2487204.85     13499875.36
      2490277.59     13499269.29      2490480.44     13497780.19
        2492675.       13498025.       2494435.5     13496126.22
       2497435.5     13497323.78      2499150.08      13496224.8
      2504409.81     13497675.44        2511025.       13496175.

Type RM Length L Ch R = 1 ,87005   ,473,473,473
BEGIN DESCRIPTION:
EIGHTEENMILE CREEK 147.0
END DESCRIPTION:
XS GIS Cut Line= 3
      2451225.01     13508875.01        2450625.       13508375.
      2449924.97     13507574.97
#Sta/Elev= 30
  4214.6   306.1  4314.2  304.47  4349.3  302.04  4475.9  300.99    4527  301.66
  4569.3  299.91  4607.2  300.06  4661.8  300.71  4802.8  298.98  4974.2  297.52
  4986.9  296.43  4992.4  292.55    4999  292.55  5000.2  291.37  5000.6  290.87
  5005.3  291.37  5031.2  297.65    5115  297.37  5150.3  297.93    5222  296.68
  5236.2  297.64  5243.8  295.05  5250.5   295.2  5258.1  292.84  5264.7  293.13
  5272.3  297.55  5300.8  298.46  5392.8  297.41  5484.9  298.17  6058.7  310.71
#Mann= 9 ,-1 , 0
  4214.6     .12       0  4475.9     .07       0  4607.2    .035       0
  4802.8     .07       0  4986.9     .12       0  5000.2     .05       0
  5005.3     .12       0    5115     .07       0  5150.3     .12       0
Bank Sta=5000.2,5005.3
XS Rating Curve= 0 ,0
Exp/Cntr=0.3,0.1

Type RM Length L Ch R = 1 ,86532   ,588,588,588
BEGIN DESCRIPTION:
EIGHTEENMILE CREEK 146.0
END DESCRIPTION:
XS GIS Cut Line= 3
        2451425.       13508375.        2450925.       13508125.
      2450124.99     13507324.99
#Sta/Elev= 30
  4436.9  305.18  4473.2  304.84  4571.1  300.24  4646.1  299.33  4884.1  298.05
  4892.5  297.55  4898.1  295.96  4920.4  295.76  4937.2  294.25  4959.6   294.5
  4965.2   293.7  4973.6  293.77  4981.9  295.61  4993.1   292.7  4999.4   292.7
  5007.3  290.23  5007.8  289.73  5012.8  290.23  5024.2  292.91  5031.3   293.5
  5038.3  295.83  5100.7  295.99  5307.8  295.62  5366.9  295.68  5462.6  295.77
  5561.6   297.6  5575.7  298.57  5618.2  298.48  5731.3  300.79  6127.3  312.03
#Mann= 7 ,-1 , 0
  4436.9     .12       0  4646.1     .07       0  5007.3     .05       0
  5012.8     .07       0  5100.7     .12       0  5307.8     .07       0
  5366.9     .12       0
Bank Sta=5007.3,5012.8
XS Rating Curve= 0 ,0
Exp/Cntr=0.3,0.1

Type RM Length L Ch R = 1 ,85944   ,300,300,300
BEGIN DESCRIPTION:
Mapping XS aef943da
END DESCRIPTION:
XS GIS Cut Line= 3
      2451407.57     13508079.64      2450825.94     13507658.61
      2450318.16     13507298.39
#Sta/Elev= 30
  4280.1  300.98    4353  298.93    4450  297.33  4493.1  297.44  4506.4  296.87
  4529.7   297.4  4678.3  295.39  4692.8  295.92  4722.2  294.91  4743.1  295.25
  4751.6   294.5  4814.2  295.44  4857.7   295.1  4893.9  294.28  4944.2  294.73
    4965  294.05  4979.7  294.72  4986.9  290.82  4991.7  287.29  4992.1  286.79
  4997.2  287.29  5001.8  287.44  5030.1  294.53  5054.8  294.02  5101.5  294.11
  5202.4  297.17    5238  297.33  5353.4  299.83  5431.2  301.64  5620.7  307.98
#Mann= 7 ,-1 , 0
  4280.1     .12       0    4353     .07       0  4857.7     .12       0
  4991.7     .05       0  4997.2     .12       0  5054.8     .07       0
  5353.4     .12       0
Bank Sta=4991.7,4997.2
XS Rating Curve= 0 ,0
Exp/Cntr=0.3,0.1

Type RM Length L Ch R = 1 ,85644   ,464,464,464
BEGIN DESCRIPTION:
EIGHTEENMILE CREEK 144.0
END DESCRIPTION:
XS GIS Cut Line= 3
      2451624.98     13508124.98        2450825.       13507375.
      2450524.97     13507224.98
#Sta/Elev= 30
  3920.1  306.34  4068.8  303.17  4097.1  301.29    4104  302.39  4111.3  301.42
  4132.3  301.86  4221.2  298.54  4365.8  296.49  4594.4  294.86  4618.8  294.38
  4716.8  294.35  4853.8  292.71  4875.2  294.53  4931.9  294.27  4946.1  292.47
  4952.9  293.48  4960.2  288.54  4967.1  288.83  4971.6  287.96    4972  287.46
  4977.2  287.96  4988.6  289.36  4995.4  289.15  5002.7  290.54  5009.6   290.1
  5013.2  292.54  5032.1  293.81  5115.8  295.93  5136.8  297.13  5352.1  302.91
#Mann= 9 ,-1 , 0
  3920.1     .12       0  4221.2     .07       0  4594.4     .12       0
  4618.8     .07       0  4716.8     .12       0  4971.6     .05       0
  4977.2     .12       0  5032.1     .07       0  5115.8     .12       0
Bank Sta=4971.6,4977.2
XS Rating Curve= 0 ,0
Exp/Cntr=0.3,0.1

Type RM Length L Ch R = 1 ,85180   ,178,178,178
BEGIN DESCRIPTION:
EIGHTEENMILE CREEK 143.0
END DESCRIPTION:
XS GIS Cut Line= 3
      2451875.02     13507875.02        2451075.       13507075.
        2450675.       13506825.
#Sta/Elev= 30
  3869.2  307.86  3917.5   306.7  4081.4  302.58  4095.5     303  4208.6  300.75
  4222.8  301.28  4359.6   297.1  4477.3  294.79  4640.9  293.75  4651.6  293.67
  4786.5  291.62    4845  291.32  4859.2  292.06  4873.3  291.21  4901.6   292.5
  4915.7  291.91  4929.9  292.76  4958.2  292.68  4972.3  292.35  4983.7   287.8
  4984.1   287.3  4989.3   287.8  5029.5  289.33    5036  292.18  5044.8  292.69
  5087.3  290.56  5193.5  294.75  5248.7  295.73  5306.6   296.9  5472.3  302.61
#Mann= 10 ,-1 , 0
  3869.2     .07       0  3917.5     .12       0  4359.6     .07       0
  4640.9     .12       0  4651.6     .07       0  4786.5     .12       0
  4983.7     .05       0  4989.3     .12       0  5193.5     .07       0
  5248.7     .12       0
Bank Sta=4983.7,4989.3
XS Rating Curve= 0 ,0
Exp/Cntr=0.3,0.1

Type RM Length L Ch R = 1 ,85002   ,749,749,749
BEGIN DESCRIPTION:
Mapping XS 7c6bfa75
END DESCRIPTION:
XS GIS Cut Line= 3
      2451785.16     13507359.15      2451077.67     13506899.06
      2450713.09     13506656.01
#Sta/Elev= 30
  4152.8  298.55  4206.5     298  4248.7  296.47  4297.5  295.72  4570.9  292.96
  4713.6  290.68  4785.2  292.23  4813.3  291.72  4849.5  292.53  4892.6  291.26
  4928.3  292.21  4973.4  292.39    4988  291.47  4993.9  287.54  4994.4  287.04
  4999.1  287.04  4999.5  287.54    5024   287.9  5034.7  291.98  5036.5  292.67
  5051.6  291.64  5066.6     293  5087.6  293.09  5096.1  293.98  5128.9  294.17
  5240.3  297.07    5319  299.96  5384.5  301.48  5391.1  302.29  5434.9   303.3
#Mann= 7 ,-1 , 0
  4152.8     .12       0  4297.5     .07       0  4570.9     .12       0
  4993.9     .05       0  4999.5     .12       0  5034.7     .07       0
  5128.9     .12       0
Bank Sta=4993.9,4999.5
XS Rating Curve= 0 ,0
Exp/Cntr=0.3,0.1

Type RM Length L Ch R = 1 ,84253   ,280,280,280
BEGIN DESCRIPTION:
EIGHTEENMILE CREEK 141.0
END DESCRIPTION:
XS GIS Cut Line= 3
      2451925.02     13507125.03        2451525.       13506625.
      2450724.96     13506274.98
#Sta/Elev= 30
  4359.6  297.69  4364.3  297.59  4501.3  296.01  4558.9  293.99  4695.8  293.41
  4850.3  290.86  4885.5  285.48  4893.5  285.51  4907.9   289.5  4922.3   288.1
  4928.7  285.82  4943.1  284.71  4949.5  282.91  4971.9  284.09  4986.3  282.97
  4992.7  284.25  4993.8  282.68  4994.3  282.18  4999.6  282.68  5008.9  284.05
  5014.4  282.87  5032.3  286.18  5037.8  284.37  5043.6  287.61  5054.5  290.13
  5236.1   290.9  5415.7  292.31  5707.5  301.77  5835.3  307.41  5873.2  307.46
#Mann= 7 ,-1 , 0
  4359.6     .12       0  4364.3     .07       0  4695.8     .12       0
  4993.8     .05       0  4999.6     .12       0  5236.1     .07       0
  5415.7     .12       0
Bank Sta=4993.8,4999.6
XS Rating Curve= 0 ,0
Exp/Cntr=0.3,0.1

Type RM Length L Ch R = 1 ,83973   ,319,319,319
BEGIN DESCRIPTION:
Mapping XS 5c5fe6da
END DESCRIPTION:
XS GIS Cut Line= 3
      2452304.79     13507083.05       2451752.7      13506494.5
      2450872.51     13506077.84
#Sta/Elev= 30
  4157.7  302.48  4715.2  292.07  4757.7   290.3  4764.6  287.91  4771.9  289.54
  4778.7  287.36  4792.9  290.45  4799.8  287.49  4807.1  289.38  4813.9  286.36
  4827.9   286.2  4863.8  286.28  4884.7   287.1  4892.1   284.8  4898.9  288.79
  4920.4  285.97  4941.4  289.34  4971.4   289.7    4977  288.53  4984.3  282.86
  4991.2   282.8  4991.7   282.3  4997.2   282.8  5028.5  285.56  5039.6  287.36
  5045.2  290.29    5264  288.88  5396.5  289.57  5526.4  291.78  5938.5  305.68
#Mann= 7 ,-1 , 0
  4157.7     .12       0  4827.9     .07       0  4863.8     .12       0
  4991.2     .05       0  4997.2     .12       0    5264     .07       0
  5396.5     .12       0
Bank Sta=4991.2,4997.2
XS Rating Curve= 0 ,0
Exp/Cntr=0.3,0.1

Type RM Length L Ch R = 1 ,83654   ,491,491,491
BEGIN DESCRIPTION:
Mapping XS ca634915
END DESCRIPTION:
XS GIS Cut Line= 3
       2452554.8     13506916.39      2451893.33     13506249.71
      2450919.67     13505822.76
#Sta/Elev= 30
    4065  304.59  4255.6  300.49    4266   300.4  4553.7  295.97  4560.8  296.69
  4758.8  290.25  4886.1  289.65  4928.5  285.19  4935.6  285.84  4942.6  288.57
  4956.8  288.84    4978   286.2  5000.9  281.53  5001.4  281.03  5006.9  281.53
  5023.5  287.82  5035.1  290.31  5057.8  288.74  5144.9  288.58  5209.8  287.14
  5242.5  288.53  5340.8     288  5354.6  287.38    5378  284.16  5395.4  284.44
  5406.8  286.94  5453.6  289.17    5702  294.45  6025.5  302.74  6067.3  303.63
#Mann= 8 ,-1 , 0
    4065     .12       0  4255.6     .07       0    4266     .12       0
  5000.9     .05       0  5006.9     .12       0  5144.9     .07       0
    5702     .12       0  6025.5     .07       0
Bank Sta=5000.9,5006.9
XS Rating Curve= 0 ,0
Exp/Cntr=0.3,0.1

Type RM Length L Ch R = 1 ,83163   ,474,474,474
BEGIN DESCRIPTION:
Mapping XS 27216d29
END DESCRIPTION:
XS GIS Cut Line= 3
      2452763.12     13506853.87      2452096.45     13505926.79
      2451195.43     13505307.01
#Sta/Elev= 30
  3841.2  305.69  4041.7  300.47  4061.5  300.14  4097.9  293.68  4139.7  294.39
  4154.4  291.71  4160.5  297.44  4175.3  298.27  4183.8  295.17  4210.9  297.66
  4338.1   295.6  4566.3  291.56  4703.3  288.89  4849.8  287.03  4871.3  283.83
  4877.4  286.16    4913  286.06  4971.9  282.77  4978.1  280.35  4978.6  279.85
  4984.1  280.35  4999.1  286.56  5070.8  286.59  5100.6  282.76  5121.5  286.31
  5166.2   284.5  5251.9  286.95  5309.6  281.93  5415.4  287.66  6076.7  297.89
#Mann= 8 ,-1 , 0
  3841.2     .12       0  4041.7     .07       0  4338.1     .12       0
  4566.3     .07       0  4703.3     .12       0  4978.1     .05       0
  4984.1     .12       0  5415.4     .07       0
Bank Sta=4978.1,4984.1
XS Rating Curve= 0 ,0
Exp/Cntr=0.3,0.1

Type RM Length L Ch R = 1 ,82689   ,223,223,223
BEGIN DESCRIPTION:
Mapping XS 4e534ab2
END DESCRIPTION:
XS GIS Cut Line= 3
      2453065.19     13506468.45      2452481.87     13505791.38
      2451478.35     13505198.63
#Sta/Elev= 30
  4089.7  306.17  4141.6  305.28  4362.4  299.37    4638  293.16  4645.6  292.84
  4652.2  289.49  4659.9  290.12  4680.7  286.53  4715.9  288.32  4730.1  290.98
  4780.6  284.53  4801.4   285.7    4808  289.14  4822.3  289.46  4934.8  287.14
    4950  286.54  4964.9  286.25  4974.7   279.5  4975.2     279  4980.7   279.5
  4991.6  281.73  5044.4  282.73  5087.9  286.33  5277.5  284.94  5318.2   285.2
  5438.4  280.85    5497  286.21  5527.7   286.8  5988.8  298.11  6148.9  302.43
#Mann= 12 ,-1 , 0
  4089.7     .07       0  4141.6     .12       0  4362.4     .07       0
  4934.8     .12       0    4950     .07       0  4974.7     .05       0
  4980.7     .07       0  5087.9     .12       0  5277.5     .07       0
  5318.2     .12       0  5527.7     .07       0  5988.8     .12       0
Bank Sta=4974.7,4980.7
XS Rating Curve= 0 ,0
Exp/Cntr=0.3,0.1

Type RM Length L Ch R = 1 ,82466   ,474,474,474
BEGIN DESCRIPTION:
EIGHTEENMILE CREEK 137.0
END DESCRIPTION:
XS GIS Cut Line= 3
      2453025.03     13505975.03        2452625.       13505625.
      2451875.01     13504975.01
#Sta/Elev= 30
  4468.5  298.34  4489.4  298.02  4567.7  295.16  4653.1  293.49  4659.8  294.05
  4702.5  291.59  4759.4  290.36  4801.2  288.36    4875  287.06  4915.1   286.4
  4929.3  284.77  4943.6  281.39  4950.2   282.2  4957.8  280.78  5013.8  280.32
  5035.7  284.97  5134.4  283.96  5205.7  285.82  5318.7  283.63  5340.5  281.55
  5375.8  279.72  5380.2  278.75  5380.7  278.25  5386.4  278.75    5425  280.65
  5461.2  286.18  5731.6  292.56  5807.8  294.45  5899.9  298.19  5992.5  299.67
#Mann= 9 ,-1 , 0
  4468.5     .07       0  4489.4     .12       0    4875     .07       0
  4957.8     .05       0  5013.8     .07       0  5375.8     .07       0
  5380.2     .07       0  5386.4     .07       0  5731.6     .12       0
Bank Sta=4957.8,5013.8
XS Rating Curve= 0 ,0
Exp/Cntr=0.3,0.1

Type RM Length L Ch R = 1 ,81992   ,446,446,446
BEGIN DESCRIPTION:
EIGHTEENMILE CREEK 136.0
END DESCRIPTION:
XS GIS Cut Line= 3
      2453074.98     13505574.96        2452875.       13505275.
        2452225.       13504975.
#Sta/Elev= 30
  4639.9  290.72    4824  285.59    4857  284.88  4964.4  282.72  4977.9  277.47
  4992.9  279.08  5032.3  279.06    5055  279.34  5099.5   277.7  5129.4  279.98
  5134.9  278.97  5152.3  279.38  5157.8   278.3  5177.2  278.05  5184.5  276.95
    5185  276.45  5190.7  276.95  5226.7  278.41  5232.2  279.65  5264.7  281.76
    5278  283.97  5295.5  282.25  5337.7   284.3  5352.8  284.89  5363.9  283.89
  5425.6  286.47  5441.9  286.43    5516  289.07  5541.5  288.76  5716.3  293.69
#Mann= 11 ,-1 , 0
  4639.9     .07       0    4824     .05       0    4857      .1       0
  5032.3     .12       0  5177.2     .07       0  5184.5     .05       0
  5190.7     .07       0  5337.7     .12       0  5425.6     .07       0
  5441.9     .12       0    5516     .07       0
Bank Sta=5184.5,5190.7
XS Rating Curve= 0 ,0
Exp/Cntr=0.3,0.1

Type RM Length L Ch R = 1 ,81546   ,453,453,453
BEGIN DESCRIPTION:
EIGHTEENMILE CREEK 135.0
END DESCRIPTION:
XS GIS Cut Line= 3
      2453474.98     13505024.99        2453075.       13504925.
      2452425.01       13504525.
#Sta/Elev= 30
  4591.9  290.44  4644.8  288.51  4680.1  287.21    4780  285.62  4816.1  284.02
  4839.3  284.54  4880.5  281.04  4898.5  280.68  4903.7  279.83  4921.7  280.15
  4966.3  276.91  4977.6  275.39  4978.1  274.89  4984.3  275.39  4986.2  276.77
  4993.9  277.28  5033.2  276.14  5039.4  278.34  5075.7  281.79  5112.4  279.66
  5127.8  281.13  5156.8  281.25  5179.9   278.2  5215.5  277.57  5280.5  280.68
  5286.4  282.42  5321.2  283.24  5378.1  284.25  5607.1  289.49  5767.4  294.69
#Mann= 8 ,-1 , 0
  4591.9     .07       0  4644.8     .05       0  4680.1     .07       0
  4966.3     .12       0  4977.6     .05       0  4984.3     .12       0
  5321.2     .07       0  5378.1     .12       0
Bank Sta=4977.6,4984.3
XS Rating Curve= 0 ,0
Exp/Cntr=0.3,0.1

Type RM Length L Ch R = 1 ,81093   ,468,468,468
BEGIN DESCRIPTION:
EIGHTEENMILE CREEK 134.0
END DESCRIPTION:
XS GIS Cut Line= 3
      2453575.03     13504675.01        2453225.       13504525.
        2452575.       13504375.
#Sta/Elev= 30
  4619.6  289.78  4652.3  289.45  4757.4  284.98  4798.7  284.54    4810  284.75
  4815.5   283.2  4833.6  283.76  4956.9     281  4978.7  279.24  4985.9  274.97
  4987.2  275.09  4991.4  275.46  4994.4  271.58  4994.9  271.08  5001.1  271.58
    5003  271.58  5010.7  275.38  5028.6  275.38    5103  277.65  5133.9  279.79
  5164.6  279.57  5174.9  275.85  5195.4  274.75  5248.4  278.41  5339.1  282.64
  5391.4  283.45    5452  284.13  5583.7  290.06  5622.7  291.05  5667.5   292.2
#Mann= 10 ,-1 , 0
  4619.6     .07       0  4798.7     .12       0  4987.2     .07       0
  4994.4     .05       0  5001.1     .07       0  5028.6     .12       0
  5133.9     .07       0  5391.4     .12       0  5583.7     .07       0
  5622.7     .12       0
Bank Sta=4994.4,5001.1
XS Rating Curve= 0 ,0
Exp/Cntr=0.3,0.1

Type RM Length L Ch R = 1 ,80625   ,284,284,284
BEGIN DESCRIPTION:
EIGHTEENMILE CREEK 133.0
END DESCRIPTION:
XS GIS Cut Line= 3
      2453725.01       13504325.        2453125.       13504125.
      2452724.98       13504175.
#Sta/Elev= 30
  4367.5  290.98  4399.1  289.31  4420.2  289.18  4616.5  281.88  4736.4   280.2
  4852.4  279.75  4915.6  278.14  4968.3  273.62  4978.9  274.64  4989.4  273.97
  4997.3  271.41  5002.5  271.41  5006.6  270.15  5007.1  269.65  5012.9  269.65
  5013.4  270.15  5020.1  272.71  5030.2  273.58  5042.8  273.74  5060.4  275.63
  5070.5  275.13  5090.7  275.77  5118.4  277.83  5123.4  277.69    5131  279.04
  5141.1  279.56  5251.9  282.55  5279.6  284.46  5322.5  284.23  5403.1  287.05
#Mann= 4 ,-1 , 0
  4367.5     .12       0  4616.5     .07       0  5006.6     .05       0
  5013.4     .07       0
Bank Sta=5006.6,5013.4
XS Rating Curve= 0 ,0
Exp/Cntr=0.3,0.1

Type RM Length L Ch R = 1 ,80341   ,598,598,598
BEGIN DESCRIPTION:
Mapping XS a8c47384
END DESCRIPTION:
XS GIS Cut Line= 3
       2453690.5     13504038.81       2453074.2     13503886.91
      2452728.48     13503791.83
#Sta/Elev= 30
  4354.6  284.65  4380.9  284.13  4422.1  282.26  4474.8  281.12  4525.1  279.98
  4554.7  279.97  4607.4  278.58  4648.6  278.16  4679.2  278.92  4689.8  278.43
  4751.6  278.32  4788.7  277.81  4821.1  277.22  4875.2  276.86  4896.9  275.58
  4933.3  275.98  4957.6  274.98  4979.9  273.01  4998.9  272.58  5005.8  268.79
  5006.3  268.29  5012.2  268.29  5012.7  268.79  5014.9   273.8    5030  279.49
  5088.9  281.38  5123.3  281.39  5133.7  281.82  5169.4  281.54  5347.9  283.62
#Mann= 7 ,-1 , 0
  4354.6     .12       0  4474.8     .07       0  4788.7     .12       0
  4821.1     .07       0  5005.8     .05       0  5012.7     .07       0
  5169.4     .12       0
Bank Sta=5005.8,5012.7
XS Rating Curve= 0 ,0
Exp/Cntr=0.3,0.1

Type RM Length L Ch R = 1 ,79743   ,458,458,458
BEGIN DESCRIPTION:
EIGHTEENMILE CREEK 131.0
END DESCRIPTION:
XS GIS Cut Line= 3
      2453775.03     13503825.03        2453425.       13503475.
      2452624.99     13502674.99
#Sta/Elev= 30
    4510   283.2    4882  276.32  4920.2  276.05  4962.6   273.7  4976.7  271.98
  4990.9  268.27  4997.1  267.55  4997.6  267.05  5005.9  267.55  5008.5  267.55
  5019.2   271.4  5047.4  271.68  5061.6  272.67  5083.1  275.87  5089.9  276.84
  5330.3  278.35  5344.4  277.96  5358.6  272.14  5370.4   271.4  5399.6  272.19
  5415.1  275.96  5457.6  277.94  5528.3  276.97  5556.6   278.1  5641.4  280.77
    5979   288.7  6009.1  288.58  6023.2  290.19  6096.2  292.93  6136.4     294
#Mann= 10 ,-1 , 0
    4510     .12       0    4882     .07       0  4997.1     .05       0
  5005.9     .07       0  5083.1     .12       0  5370.4      .1       0
  5399.6     .12       0  5556.6     .07       0    5979     .12       0
  6096.2     .07       0
Bank Sta=4997.1,5005.9
XS Rating Curve= 0 ,0
Exp/Cntr=0.3,0.1

Type RM Length L Ch R = 1 ,79285   ,594,594,594
BEGIN DESCRIPTION:
Mapping XS a93208ce
END DESCRIPTION:
XS GIS Cut Line= 3
      2454200.65     13503708.07      2453721.45     13503187.21
      2452903.75     13502567.43
#Sta/Elev= 30
  4284.6  286.13  4609.3  282.44  4835.6  278.49  4920.6  276.56    4949   273.3
  4955.8  271.02  4960.8  270.79  4977.4  268.99  4984.2  267.38    4986  265.46
  4986.5  264.96  4994.9  265.46    5013  269.99  5034.6  271.97  5132.4  275.08
  5184.4  271.66  5208.5  271.65  5253.1  268.82  5269.7  269.17  5276.5  272.94
  5290.5  275.56  5373.9  275.27  5390.4  274.52    5434  276.18  5463.1  272.96
    5484  275.85  5504.8  275.08  5569.3  277.25  5733.6  278.04  6018.4  287.79
#Mann= 8 ,-1 , 0
  4284.6     .12       0  4960.8     .07       0    4986     .05       0
  4994.9     .07       0  5132.4     .12       0  5208.5      .1       0
  5253.1     .12       0  5373.9     .07       0
Bank Sta=4986,4994.9
XS Rating Curve= 0 ,0
Exp/Cntr=0.3,0.1

Type RM Length L Ch R = 1 ,78691   ,926,926,926
BEGIN DESCRIPTION:
Mapping XS bf02b964
END DESCRIPTION:
XS GIS Cut Line= 4
      2454783.92      13503452.8      2453976.66     13502676.79
      2453398.54     13502567.42      2453070.39     13502010.09
#Sta/Elev= 30
  3675.3  279.09  3681.1  278.97  3744.6  279.17  4065.2   276.8  4401.4  274.27
  4884.3  275.87  4959.6  274.22  4975.3  264.55  4975.8  264.05  4984.5  264.55
  5010.5  268.16  5051.5  265.54  5091.9  270.29  5112.2  269.51  5154.1  276.44
  5173.3  275.54    5214   266.7  5253.6  268.08  5353.1  274.41  5460.5  276.17
  5476.2  273.83  5511.9  276.86  5540.6  276.63  5548.7  271.53  5650.1  278.31
  5693.2  279.28    5812  281.44  5854.9  285.53  5909.4  281.98  6030.2  286.99
#Mann= 13 ,-1 , 0
  3675.3     .12       0  3681.1     .07       0  3744.6     .12       0
  4065.2     .07       0  4975.3     .05       0  4984.5     .07       0
  5154.1     .12       0  5253.6     .07       0  5353.1     .12       0
  5511.9     .07       0  5650.1     .12       0  5693.2     .07       0
  5909.4     .05       0
Bank Sta=4975.3,4984.5
XS Rating Curve= 0 ,0
Exp/Cntr=0.3,0.1

Type RM Length L Ch R = 1 ,77765   ,453,453,453
BEGIN DESCRIPTION:
Mapping XS 6f730117
END DESCRIPTION:
XS GIS Cut Line= 3
      2454966.26     13503468.49      2454309.99     13502473.67
      2454263.12     13501385.16
#Sta/Elev= 30
  3609.6  280.14  3935.3  275.03  3942.5  275.05  4263.1  273.36  4620.5  273.15
  4814.8   272.8  4880.1  270.62  4954.4  270.07  4970.2  267.57  4995.5  260.26
    4996  259.76    5005  260.26  5033.7  263.59  5040.3  265.75  5070.3  265.99
  5128.9  270.46  5140.4  269.06  5150.4  266.14  5220.4  270.62  5319.4  272.94
  5450.7  274.31  5480.7   278.7  5490.7  277.67  5502.1  273.12  5560.8  272.84
  5580.8  278.47  5610.8  276.67  5733.5  278.45    5781  280.93  5890.9  283.57
#Mann= 11 ,-1 , 0
  3609.6     .07       0  3935.3     .12       0  3942.5     .07       0
  4263.1     .12       0  4620.5     .07       0  4814.8     .12       0
  4954.4     .07       0  4995.5     .05       0    5005     .07       0
  5128.9     .12       0  5319.4     .07       0
Bank Sta=4995.5,5005
XS Rating Curve= 0 ,0
Exp/Cntr=0.3,0.1

Type RM Length L Ch R = 1 ,77312   ,935,935,935
BEGIN DESCRIPTION:
Mapping XS 3e2a7f79
END DESCRIPTION:
XS GIS Cut Line= 3
      2455106.87     13503557.01      2454763.12     13502390.33
      2454627.78      13501479.4
#Sta/Elev= 30
  3616.6  282.86  3629.1  281.83  3660.4  281.82  3733.2  279.88  3879.3  276.65
  4251.2  271.61  4285.9  270.12  4358.9  270.88  4489.6  269.35  4765.4  270.02
  4786.3  268.81  4868.6  269.84  4929.2  269.43  4949.5  267.23  4969.7  261.55
  4987.5  260.36  4987.8  259.26  4988.3  258.76  4997.3  259.26  5010.1  262.96
  5050.6  264.96    5091  268.38  5131.4  269.16  5171.9  268.43  5265.1  271.87
  5444.8  275.96  5515.6  279.13  5525.7  278.44  5568.4  279.61  5753.8  285.74
#Mann= 6 ,-1 , 0
  3616.6     .12       0  3733.2     .07       0  4251.2     .12       0
  4987.8     .05       0  4997.3     .12       0  5568.4     .07       0
Bank Sta=4987.8,4997.3
XS Rating Curve= 0 ,0
Exp/Cntr=0.3,0.1

Type RM Length L Ch R = 1 ,76377   ,568,568,568
BEGIN DESCRIPTION:
Mapping XS c5cd6faf
END DESCRIPTION:
XS GIS Cut Line= 4
      2455336.05     13503635.16      2455023.54     13502713.25
       2455377.7     13502520.54      2455190.21     13501442.46
#Sta/Elev= 30
  3797.3  285.63  4063.2  278.61  4643.2  269.13    4689  268.06  4705.5  264.27
  4715.1  264.23  4746.5  268.16    4794  268.15  4837.7  267.31  4843.4  264.96
  4852.1  264.61  4881.3  265.31    4909  262.71    4925  264.75  4931.8  267.06
  4954.5  267.13  4990.6  264.89  5000.2  261.83  5007.6  258.69  5008.1  258.19
  5017.2  258.69  5028.6  260.39  5072.3  262.75  5088.4  266.64  5094.1  266.05
  5102.5  268.12  5148.1  269.18  5311.5  267.74    5545  269.17  6268.2   278.2
#Mann= 6 ,-1 , 0
  3797.3     .12       0  4063.2     .07       0  4643.2     .12       0
  5000.2     .07       0  5007.6     .05       0  5017.2     .07       0
Bank Sta=5007.6,5017.2
XS Rating Curve= 0 ,0
Exp/Cntr=0.3,0.1

Type RM Length L Ch R = 1 ,75809   ,571,571,571
BEGIN DESCRIPTION:
Mapping XS 9b515026
END DESCRIPTION:
XS GIS Cut Line= 3
      2455523.54     13503676.77      2455622.49     13502921.58
       2455299.8     13501292.48
#Sta/Elev= 30
  4190.9  287.41  4676.8     276  4797.8   272.1    4818  269.74  4828.1  271.19
  4838.2  270.78  4854.8  265.08  4859.9  269.49  4878.5  262.85  4888.6  262.75
  4898.7   264.3  4908.8  263.39  4928.6  264.45  4933.7  266.62  4952.5  266.18
  4959.3  265.81  4979.6   260.1  5005.2  258.61  5005.7  258.11  5015.2  258.61
  5040.8  259.19  5061.2  262.96  5067.3  265.11  5083.4  266.21  5379.7  268.02
  5516.8  267.37  5733.1  268.18  6274.3  273.95    6417  276.33  6613.3   281.4
#Mann= 5 ,-1 , 0
  4190.9     .07       0  5005.2     .05       0  5015.2     .07       0
  5083.4     .12       0  5516.8     .07       0
Bank Sta=5005.2,5015.2
XS Rating Curve= 0 ,0
Exp/Cntr=0.3,0.1

Type RM Length L Ch R = 1 ,75238   ,534,534,534
BEGIN DESCRIPTION:
Mapping XS d650c8d3
END DESCRIPTION:
XS GIS Cut Line= 3
      2456299.58     13503536.19      2456158.95     13502780.96
      2455471.44     13501333.01
#Sta/Elev= 30
  4201.8  283.28  4304.2   282.9  4325.1  281.68    4437  280.71  4620.1  277.55
  4773.9  273.63  4843.8  271.36  4965.3  265.03    4970  265.24  4976.6  262.83
  4986.5  256.65  4993.7  255.19  4994.2  254.69  5003.8  255.19  5009.2  256.78
  5037.5  259.58  5065.8  261.23    5083  260.71  5105.7  263.31    5134  264.05
  5151.1  265.74  5330.9  265.76  5338.5  264.57  5622.3  267.09  5917.6  267.84
  6036.9  270.29  6094.7  270.12  6292.4  273.17    6498  279.01  6572.9  281.01
#Mann= 6 ,-1 , 0
  4201.8     .07       0  4773.9     .12       0  4965.3     .07       0
  4993.7     .05       0  5003.8     .07       0    6498     .12       0
Bank Sta=4993.7,5003.8
XS Rating Curve= 0 ,0
Exp/Cntr=0.3,0.1

Type RM Length L Ch R = 1 ,74704   ,203,203,203
BEGIN DESCRIPTION:
EIGHTEENMILE CREEK 123.0
END DESCRIPTION:
XS GIS Cut Line= 3
        2456575.     13502824.99        2456625.       13502575.
      2456174.99     13501824.99
#Sta/Elev= 30
  4740.8  269.61  4812.2  267.77  4824.2  266.71    4853  264.55  4868.3   265.9
  4893.8  264.63  4914.2  263.31  4924.4  260.68  4933.2  259.78  5009.3  256.18
    5014  253.38  5014.5  252.88  5024.2  253.38  5030.7  257.74  5040.4  262.17
  5046.3  259.31    5054  262.95    5089  265.13  5162.9  262.84  5205.7  262.43
  5279.5  262.59  5438.9  265.05    5470  263.68  5475.8     264  5485.5  262.81
  5660.5  265.22  5703.2  265.03    5746  266.47  5786.9  266.61  5870.4  267.74
#Mann= 6 ,-1 , 0
  4740.8     .07       0  4824.2     .12       0  4933.2     .07       0
    5014     .05       0  5024.2     .07       0  5786.9     .12       0
Bank Sta=5014,5024.2
XS Rating Curve= 0 ,0
Exp/Cntr=0.3,0.1

Type RM Length L Ch R = 1 ,74501   ,696,696,696
BEGIN DESCRIPTION:
EIGHTEENMILE CREEK 122.0
END DESCRIPTION:
XS GIS Cut Line= 3
       2456850.8     13502866.11      2456809.78     13502524.46
      2456332.56     13501485.85
#Sta/Elev= 30
  4655.9  270.13  4718.5  268.62  4777.5   267.3  4850.7  265.38    4929   262.2
    4939  259.95  4991.1  255.28  4991.6  254.78  5001.4  255.28  5010.4  256.24
  5025.2  256.42  5065.4  262.62  5076.6  261.36  5094.1  261.19  5099.6  258.34
  5117.1   260.2  5131.5  256.87  5140.1   260.7  5145.6  260.06  5163.1  261.12
    5243  262.04  5386.4  262.66  5439.6  260.27  5529.8  263.32  5547.3  262.35
  5552.8  262.81  5570.2  261.87  5621.7   261.3    5811  264.96    6143  267.82
#Mann= 6 ,-1 , 0
  4655.9     .05       0  4718.5     .07       0  4777.5     .12       0
  4850.7     .07       0  4991.1     .05       0  5001.4     .07       0
Bank Sta=4991.1,5001.4
XS Rating Curve= 0 ,0
Exp/Cntr=0.3,0.1

Type RM Length L Ch R = 1 ,73805   ,418,418,418
BEGIN DESCRIPTION:
EIGHTEENMILE CREEK 121.0
END DESCRIPTION:
XS GIS Cut Line= 3
      2457424.99     13502624.98        2457275.       13502075.
      2456869.51     13501151.03
#Sta/Elev= 30
  4423.2  267.74  4514.7  265.71  4599.4  265.53  4728.1  263.91  4827.4   262.6
  4920.7   259.7  4941.4  257.96  4962.2  254.12    4976   252.9  4982.9  253.15
  4985.4  252.48  4985.9  251.98  4995.5  251.98    4996  252.48  5015.1  254.38
    5031  254.96  5146.2  255.46  5252.2  258.35  5257.7     259  5275.6  259.24
    5299  260.47  5374.5  259.93  5408.8  260.97  5551.1  261.04  5601.1  260.46
  5653.3  261.32  5728.9  263.56  5757.7  264.99  5846.8   266.8  6002.3  270.88
#Mann= 6 ,-1 , 0
  4423.2     .05       0  4728.1     .07       0  4985.4     .05       0
    4996     .07       0  5551.1     .05       0  5846.8     .07       0
Bank Sta=4985.4,4996
XS Rating Curve= 0 ,0
Exp/Cntr=0.3,0.1

Type RM Length L Ch R = 1 ,73387   ,467,467,467
BEGIN DESCRIPTION:
EIGHTEENMILE CREEK 120.0
END DESCRIPTION:
XS GIS Cut Line= 3
        2457575.     13502725.02        2457475.       13501725.
        2457275.     13501074.98
#Sta/Elev= 30
    3999  270.17  4152.3   266.2  4260.3   265.1  4313.2  263.74  4531.7  260.27
  4712.6  259.53  4755.3  260.34  4833.2  255.94  4855.8  256.84  4913.6  255.76
  4943.7  253.22  4956.3  253.54  4973.9  251.81  4983.9  252.19    4996  251.22
  4996.5  250.72    5007  251.22  5020.4   254.7  5045.9  253.55  5058.3  253.96
  5077.2  256.67  5098.2   256.7  5118.4  258.03  5123.7  257.43    5140  259.39
  5325.1  263.39  5466.3  265.27    5635  269.68  5662.5  271.85  5684.1  272.29
#Mann= 4 ,-1 , 0
    3999     .05       0  4313.2     .07       0    4996     .05       0
    5007     .07       0
Bank Sta=4996,5007
XS Rating Curve= 0 ,0
Exp/Cntr=0.3,0.1

Type RM Length L Ch R = 1 ,72920   ,735,735,735
BEGIN DESCRIPTION:
EIGHTEENMILE CREEK 119.0
END DESCRIPTION:
XS GIS Cut Line= 3
        2457825.     13502524.96        2457925.       13501775.
      2457725.01     13501225.03
#Sta/Elev= 30
  4243.3  265.98  4394.6  260.98  4460.2  259.87  4525.7  258.42  4545.9  258.98
  4616.5   252.4  4655.6  253.06  4660.7  251.96  4677.1   253.3  4697.2  258.04
  4738.9  257.82    4788  253.82  4818.3  257.44  4848.6   258.3  4890.2  255.61
  4958.3  255.31  4969.6  253.32  5002.6   251.5  5009.7  249.68  5010.2  249.18
  5020.7  249.68  5031.8  251.87    5085  252.08  5101.7  255.33    5107  254.39
  5126.9  257.18  5132.2  255.98  5170.2  261.21    5351   261.8  5585.1  264.94
#Mann= 4 ,-1 , 0
  4243.3     .05       0  4460.2     .07       0  5009.7     .05       0
  5020.7     .07       0
Bank Sta=5009.7,5020.7
XS Rating Curve= 0 ,0
Exp/Cntr=0.3,0.1

Type RM Length L Ch R = 1 ,72185   ,413,413,413
BEGIN DESCRIPTION:
Mapping XS cdcde2cd
END DESCRIPTION:
XS GIS Cut Line= 3
      2458179.79     13502895.51      2458242.29     13502015.33
      2457945.77     13501078.95
#Sta/Elev= 30
  4277.8  273.26    4338  272.53  4408.6  271.48  4508.9  267.89  4595.9  266.27
  4649.2  263.71  4816.6  258.95    4940  255.32    4960  251.36  4990.9  250.48
  4994.6  246.58  4995.1  246.08  5005.7  246.58  5020.2  249.28  5050.2  251.62
  5100.4  252.54  5120.4  253.78  5126.7  255.61  5150.5  256.31  5268.9  256.85
  5485.7  260.34  5570.1  259.52  5590.6  260.47  5602.4  258.77  5622.1  258.58
  5661.7  260.93  5699.3  260.33  5957.6  264.42  6097.3  265.45  6142.4  267.02
#Mann= 6 ,-1 , 0
  4277.8     .05       0    4338     .07       0  4595.9     .12       0
  4816.6     .07       0  4994.6     .05       0  5005.7     .07       0
Bank Sta=4994.6,5005.7
XS Rating Curve= 0 ,0
Exp/Cntr=0.3,0.1

Type RM Length L Ch R = 1 ,71772   ,259,259,259
BEGIN DESCRIPTION:
Mapping XS c8281514
END DESCRIPTION:
XS GIS Cut Line= 3
      2458487.09     13502812.17      2458612.08     13502072.63
      2458211.04     13501161.18
#Sta/Elev= 30
  4197.1  272.88  4255.1  272.31  4625.1  259.34  4695.4  255.85  4731.7  252.58
  4755.9  251.61  4801.7  254.97  4876.7  255.29  4883.9   252.7    4894   251.9
  4924.4  252.29  4935.7  251.45  4951.1  249.48  4956.6  249.96  4988.2  248.57
  4992.2   246.1  4992.7   245.6  5003.4   246.1    5021  249.46  5026.6  251.35
  5032.1  250.87    5050   256.7  5119.3  256.33  5381.5  259.32    5395  258.87
    5458  258.78  5572.9  260.24  5596.2  259.65  5799.3  262.62  5942.9  263.64
#Mann= 7 ,-1 , 0
  4197.1     .07       0  4625.1     .12       0  4801.7     .07       0
  4935.7     .05       0  4992.2     .05       0  5003.4     .05       0
    5395     .07       0
Bank Sta=4992.2,5003.4
XS Rating Curve= 0 ,0
Exp/Cntr=0.3,0.1

Type RM Length L Ch R = 1 ,71513   ,812,812,812
BEGIN DESCRIPTION:
Mapping XS 78daa7d9
END DESCRIPTION:
XS GIS Cut Line= 4
      2458497.51     13502890.31      2458731.87     13502296.58
      2458882.91     13501984.08      2458356.85     13501051.75
#Sta/Elev= 30
  4238.4  272.14  4296.1  272.72  4373.1  272.28    4434  269.76  4493.5  268.78
  4502.1  267.98  4781.7  259.36  4818.2  257.04    4828  255.56  4874.9   250.7
  4889.6  250.01    4946  250.38  4978.4  248.39  4985.6  245.37  4986.1  244.87
  4996.8  245.37  5000.6   247.3  5022.9  250.44  5030.8  252.64  5036.4  255.59
  5053.4  257.29  5098.6  255.99  5186.1  255.26  5250.8  254.44  5331.6  255.94
  5584.5  257.19  6118.3  261.22  6189.6  262.67  6227.1  262.41  6294.3  264.13
#Mann= 6 ,-1 , 0
  4238.4     .07       0    4828     .12       0  4985.6     .05       0
  4996.8     .12       0  5186.1     .05       0  5584.5     .07       0
Bank Sta=4985.6,4996.8
XS Rating Curve= 0 ,0
Exp/Cntr=0.3,0.1

Type RM Length L Ch R = 1 ,70701   ,819,819,819
BEGIN DESCRIPTION:
EIGHTEENMILE CREEK 115.0
END DESCRIPTION:
XS GIS Cut Line= 3
      2460025.04     13502475.03        2459425.       13501925.
      2458524.99     13501024.99
#Sta/Elev= 30
  4181.2  267.19  4443.7  258.52  4513.9  256.36  4627.4  255.98  4705.1  254.18
    4776   256.6  4835.3  256.06  4846.3  255.58  4853.7  252.51  4888.8  249.34
  4917.2   247.9  4924.6  249.48  4931.4  247.21    4953   246.5  4981.3  246.97
  4998.7  245.46  5001.8  242.99  5002.3  242.49  5016.8  242.99  5023.5  243.51
  5051.8  252.16  5065.9  253.74  5099.6  253.82  5136.6  252.39  5546.7  254.53
    5674  253.33  5787.1  256.39  5882.4  256.84  6241.8  262.93    6268  263.52
#Mann= 8 ,-1 , 0
  4181.2     .07       0  4443.7     .05       0  4835.3     .07       0
  5001.8     .05       0  5016.8     .07       0  5099.6     .12       0
  5882.4     .07       0  6241.8     .05       0
Bank Sta=5001.8,5016.8
XS Rating Curve= 0 ,0
Exp/Cntr=0.3,0.1

Type RM Length L Ch R = 1 ,69882   ,676,676,676
BEGIN DESCRIPTION:
Mapping XS d210604d
END DESCRIPTION:
XS GIS Cut Line= 3
      2460320.42     13502327.86      2459757.91     13501400.75
      2458731.85     13500687.19
#Sta/Elev= 30
  3570.5  265.47  3860.4   264.1  4029.1  260.77  4114.4   257.4  4638.2  252.14
  4755.6  252.33  4776.5  250.27  4841.2  246.82  4848.1  248.39  4854.1  247.68
  4862.9  249.03    4869  248.33  4883.9  249.66    4901  249.34  4955.4  248.92
  4985.1  244.22  4991.2  244.13  5004.5  240.77    5005  240.27  5019.8  240.77
  5048.2  244.37  5062.8  248.12  5071.5  252.92  5077.6   253.6  5206.6  258.26
  5279.7  259.56  5302.9   258.7  5459.1   258.9  5593.8  260.91  5904.7  264.54
#Mann= 7 ,-1 , 0
  3570.5     .05       0  4854.1     .07       0    4901     .12       0
  5004.5     .05       0  5019.8     .12       0  5302.9     .07       0
  5593.8     .05       0
Bank Sta=5004.5,5019.8
XS Rating Curve= 0 ,0
Exp/Cntr=0.3,0.1

Type RM Length L Ch R = 1 ,69206   ,560,560,560
BEGIN DESCRIPTION:
Mapping XS a4855934
END DESCRIPTION:
XS GIS Cut Line= 3
      2460836.04     13501973.68      2460028.74     13500864.29
      2458862.05     13500353.86
#Sta/Elev= 30
  3595.3  268.43  3638.3  268.48  3800.2  263.94  3832.1   263.1  3944.9  261.57
  3956.6  261.52  4036.7  260.35  4205.7  258.71  4302.4  257.33  4472.8  256.84
  4933.4  249.78  4941.7  249.06  4966.3  238.22  4969.6  238.14  4970.1  237.64
  4985.3  238.14  4993.2  241.13  5015.1  244.25  5058.7  244.25  5091.5  246.69
  5141.3  245.75  5189.7  246.29  5244.3  251.36  5342.5  251.83    5408  256.83
    5478  259.76  5758.4   262.1  6199.9  269.74  6240.2  269.61  6240.8  269.61
#Mann= 15 ,-1 , 0
  3595.3     .05       0  3800.2     .07       0  3832.1     .05       0
  3944.9     .07       0  3956.6    .035       0  4036.7     .07       0
  4205.7     .12       0  4302.4     .05       0  4472.8     .07       0
  4969.6     .05       0  4985.3     .07       0  5141.3     .12       0
  5758.4     .05       0  6199.9     .07       0  6240.2     .05       0
Bank Sta=4969.6,4985.3
XS Rating Curve= 0 ,0
Exp/Cntr=0.3,0.1

Type RM Length L Ch R = 1 ,68646   ,398,398,398
BEGIN DESCRIPTION:
Mapping XS d80fbcc6
END DESCRIPTION:
XS GIS Cut Line= 3
      2461018.33     13501900.76      2460414.16     13500489.29
      2459358.39     13499854.79
#Sta/Elev= 30
  3243.3  272.15    3245   272.1  3255.2  271.97  3668.3  261.72  3798.1  258.66
  3906.6  256.74  4222.8  253.43  4329.7  253.17  4424.3  253.22  4636.6  248.49
  4707.2  243.57  4765.4  248.12  4817.3  248.48  4855.7   244.4    4941  245.25
  4992.2  240.39  4999.8  237.17  5000.3  236.67  5015.6  237.17  5022.7  243.11
    5066  241.71    5116  248.55  5124.3   251.4  5130.1   249.4  5139.3   253.4
    5168  254.65  5501.2  265.81  5876.3  270.88  5957.4  271.61  6010.4  272.15
#Mann= 14 ,-1 , 0
  3243.3    .063       0    3245    .035       0  3255.2     .05       0
  3668.3    .035       0  3798.1     .07       0  3906.6     .05       0
  4222.8     .07       0  4329.7     .12       0  4855.7      .1       0
  4999.8     .05       0  5015.6      .1       0    5168     .12       0
  5876.3     .07       0  5957.4     .05       0
Bank Sta=4999.8,5015.6
XS Rating Curve= 0 ,0
Exp/Cntr=0.3,0.1

Type RM Length L Ch R = 1 ,68248   ,310,310,310
BEGIN DESCRIPTION:
Mapping XS 35925f01
END DESCRIPTION:
XS GIS Cut Line= 3
      2461132.92      13501853.9      2460570.41     13500208.04
      2459628.82     13499604.59
#Sta/Elev= 30
  3240.3  274.29  3328.1  271.57  3513.9  266.15  3693.6  261.94  3725.3  262.16
  3867.8  257.23  4149.6  253.21  4438.2  252.24  4655.2  248.29  4728.7   249.2
  4796.6  247.73  4890.6  241.75  4921.9  243.22  4968.5  240.96  4978.6  239.78
  4985.3  236.51  4985.8  236.01  5001.2  236.51  5008.5  239.11  5014.4  238.99
  5029.6  241.32  5044.8  245.36    5066  247.83  5274.8  254.51  5326.3  257.95
  5449.3  258.06  5492.9  259.74  5592.7  260.41  5746.2  263.74    6098  268.22
#Mann= 6 ,-1 , 0
  3240.3    .035       0  3328.1     .05       0  4438.2     .12       0
  4968.5      .1       0  4985.3     .05       0  5001.2     .12       0
Bank Sta=4985.3,5001.2
XS Rating Curve= 0 ,0
Exp/Cntr=0.3,0.1

Type RM Length L Ch R = 1 ,67938   ,379,379,379
BEGIN DESCRIPTION:
EIGHTEENMILE CREEK 110.0
END DESCRIPTION:
XS GIS Cut Line= 3
      2461125.01     13501275.05        2460825.       13500075.
      2460474.99     13499674.99
#Sta/Elev= 30
    3763  259.09  3855.8  255.36  3868.7   255.8  3987.2  253.28  4288.7  252.47
  4371.2  251.33  4433.1  252.07  4546.4  250.81  4610.9  248.07  4656.9  247.46
  4729.4  246.79  4752.6  247.92  4822.2  246.17  4899.5  247.69  4940.7  246.46
  4948.4  243.19  4963.9  240.71  4976.8  237.66  4981.7  235.39  4982.2  234.89
  4997.7  235.39  5003.3   235.7  5007.1  238.05  5017.8  238.66  5056.5  242.17
  5084.9  243.12  5134.3  248.76  5368.7  253.99  5481.7  254.71  5531.5  256.67
#Mann= 7 ,-1 , 0
    3763     .05       0  4656.9     .07       0  4822.2     .12       0
  4963.9      .1       0  4981.7     .05       0  4997.7      .1       0
  5017.8     .12       0
Bank Sta=4981.7,4997.7
XS Rating Curve= 0 ,0
Exp/Cntr=0.3,0.1

Type RM Length L Ch R = 1 ,67559   ,642,642,642
BEGIN DESCRIPTION:
Mapping XS c6321546
END DESCRIPTION:
XS GIS Cut Line= 4
       2461521.8     13501524.03      2461193.68     13499997.97
      2461094.72      13499826.1      2460485.35     13499503.18
#Sta/Elev= 30
  3354.6  268.89  3415.4  268.24  3435.4  265.29  3466.1  267.15  3496.8  266.46
  3553.3  261.72    3613  259.07  3905.9  251.72  4125.1  251.65  4325.3  247.02
  4452.5   246.8  4486.4  246.56  4666.3  245.01  4683.3  246.12  4765.1  241.09
  4789.7  241.52    4847  242.62  4889.2  242.46  4930.5  238.96  4966.9  239.08
  4996.3  234.39  4996.8  233.89  5012.3  234.39  5020.1  238.25  5063.2  241.35
    5079  248.01    5101  249.44  5439.2  252.83  5678.1  255.78  5803.5  258.66
#Mann= 12 ,-1 , 0
  3354.6    .035       0    3613     .05       0  4452.5     .12       0
  4486.4     .05       0  4666.3     .12       0  4789.7     .07       0
    4847      .1       0  4996.3     .05       0  5012.3      .1       0
    5101     .12       0  5439.2     .07       0  5678.1     .12       0
Bank Sta=4996.3,5012.3
XS Rating Curve= 0 ,0
Exp/Cntr=0.3,0.1

Type RM Length L Ch R = 1 ,66917   ,427,427,427
BEGIN DESCRIPTION:
Mapping XS 2a5973a9
END DESCRIPTION:
XS GIS Cut Line= 4
      2462084.31     13501487.58      2461704.09     13500211.52
      2461672.84     13500008.39      2460559.15     13499446.34
#Sta/Elev= 30
  3581.4  265.79  3980.8  256.09  4022.3  251.67  4121.8  252.84  4241.5  252.78
  4456.9  248.67  4578.5   247.4  4606.7  244.09  4627.5   246.2  4682.3  241.96
    4783  238.58  4794.5  241.61  4815.4  242.96  4859.8  238.28    4878  244.59
  4915.4  239.69  4937.2   237.3  4970.1  237.63  4982.3  235.42  4982.8  234.92
  4998.4  235.42  5005.5  237.49  5061.1  240.77  5117.6  242.33    5252  242.38
  5383.3  246.01  5781.6  252.48  6040.6  253.61  6270.9  255.98  6365.9  258.24
#Mann= 12 ,-1 , 0
  3581.4     .05       0  3980.8     .07       0  4121.8    .035       0
  4456.9     .05       0  4578.5     .12       0  4682.3     .05       0
  4915.4     .12       0  4982.3     .05       0  4998.4     .12       0
  5383.3     .12       0  6040.6     .07       0  6270.9     .12       0
Bank Sta=4982.3,4998.4
XS Rating Curve= 0 ,0
Exp/Cntr=0.3,0.1

Type RM Length L Ch R = 1 ,66490   ,337,337,337
BEGIN DESCRIPTION:
Mapping XS 6deefaa4
END DESCRIPTION:
XS GIS Cut Line= 3
      2463058.28     13500711.53      2462110.34     13499930.27
      2460679.01     13499451.42
#Sta/Elev= 30
  3628.7  267.77  3756.5  266.24  3862.6  262.58  4053.4  263.65  4132.9  264.31
  4294.6  263.88  4344.4  262.25  4452.3  255.29  4488.2  255.79  4600.1  248.54
  4729.8  243.06  4826.2  243.65  4883.8  241.94  4912.9  243.77  4957.7  244.41
  4978.7  235.08  4991.6  233.78  4992.1  233.28  5008.1  233.78  5010.3  236.16
  5015.6   235.9  5052.5   238.8    5105   238.5  5148.7  240.61  5189.6  244.56
  5379.4  245.38  5590.3  250.27  6204.9  254.18  6338.7  254.74  6366.4  255.55
#Mann= 15 ,-1 , 0
  3628.7     .07       0  3862.6     .05       0  4053.4     .07       0
  4132.9     .05       0  4294.6     .07       0  4344.4    .035       0
  4600.1     .05       0  4826.2     .07       0  4912.9      .1       0
  4991.6     .05       0  5008.1      .1       0  5015.6     .07       0
  5148.7     .12       0  6204.9     .07       0  6338.7     .12       0
Bank Sta=4991.6,5008.1
XS Rating Curve= 0 ,0
Exp/Cntr=0.3,0.1

Type RM Length L Ch R = 1 ,66153   ,577,577,577
BEGIN DESCRIPTION:
Mapping XS e22347d9
END DESCRIPTION:
XS GIS Cut Line= 3
      2462959.34     13500159.46      2462136.38     13499607.35
      2460668.84     13499383.57
#Sta/Elev= 30
  4013.3  271.17  4177.1  270.44  4274.2  267.31  4361.9  264.24  4423.5  259.79
  4465.6  260.23  4501.6  256.16  4546.8   253.6  4622.7  248.91  4717.7  243.56
  4789.7  242.22  4826.9  243.18  4849.4  243.35  4885.5  237.44  4916.5  237.67
  4963.7  236.69  4978.7  235.09  4985.5   232.8    4986   232.3    5002   232.8
  5002.1  236.19    5036  234.41  5075.1  236.82  5096.7  240.96  5128.3  243.29
  5400.2  247.19  5453.5  246.72  5712.6  251.93  5895.9  251.07  6488.8  255.89
#Mann= 12 ,-1 , 0
  4013.3     .05       0  4177.1     .07       0  4274.2     .05       0
  4361.9    .035       0  4546.8     .07       0  4622.7     .12       0
  4826.9     .07       0  4916.5      .1       0  4985.5     .05       0
    5002      .1       0  5075.1     .07       0  5128.3     .12       0
Bank Sta=4985.5,5002
XS Rating Curve= 0 ,0
Exp/Cntr=0.3,0.1
