--- HOOSIER CREEK.prj (project) ---

Proj Title=HOOSIER CREEK Base Level Engineering
Current Plan=p01
Default Exp/Contr=0.3,0.1
English Units
Geom File=g01
Flow File=f01
Plan File=p01
Y Axis Title=Elevation
X Axis Title(PF)=Main Channel Distance
X Axis Title(XS)=Station
BEGIN DESCRIPTION:
HOOSIER CREEK
END DESCRIPTION:
DSS Export Rating Curves= 0
DSS Export Rating Curve Sorted= 0
DSS Export Volume Flow Curves= 0
DXF OffsetX= 0
DXF OffsetY= 0
DXF ScaleX= 1
DXF ScaleY= 10

--- HOOSIER CREEK.p01 (plan) ---

Plan Title=Multiple Run
Program Version=4.10
Short Identifier=Multiple
Geom File=g01
Flow File=f01
Subcritical Flow
K Sum by GR= 0
Std Step Tol= 0.01
Critical Tol= 0.01
Num of Std Step Trials= 20
Max Error Tol= 0.3
Flow Tol Ratio= 0.001
Split Flow NTrial= 30
Split Flow Tol= 0.02
Split Flow Ratio= 0.02
Log Output Level= 0
Friction Slope Method= 1
Unsteady Friction Slope Method= 2
Unsteady Bridges Friction Slope Method= 1
Parabolic Critical Depth
Global Vel Dist= 1 , 1 , 1
Global Log Level= 0
CheckData=True
Encroach Param=-1 ,0,0, 0
BEGIN DESCRIPTION:
Multiple Run
END DESCRIPTION:
Computation Interval=1HOUR
Output Interval=1HOUR
Run HTab= 0
Run UNet= 0
Run PostProcess= 0
Run WQNet= 0
UNET Theta= 1
UNET Theta Warmup= 1
UNET ZTol= 0.02
UNET ZSATol= 0.05
UNET MxIter= 20
UNET MaxInSteps= 0
UNET DtIC= 0
UNET DtMin= 0
UNET MaxCRTS= 20
UNET WFStab= 2
UNET SFStab= 1
UNET WFX= 1
UNET SFX= 1
UNET DSS MLevel= 4
UNET DZMax Abort= 100
UNET Convert EG Bridges= 0
UNET Use Existing IB Tables=-1
UNET Froude Reduction=False
UNET Froude Limit= 1
UNET Froude Power= 10
UNET Time Slicing=0,0, 5
UNET Junction Losses=0
Instantaneous Interval=1HOUR
Write IC File= 0
Write IC File at Sim End=0
Echo Input=False
Echo Parameters=False
Echo Output=False
Write Detailed= 0
WQ AD Non Conservative
WQ ULTIMATE=-1
WQ Max Comp Step=1HOUR
WQ Output Interval=15MIN
WQ Output Selected Increments= 0
WQ Output face flow=0
WQ Output face velocity=0
WQ Output face area=0
WQ Output face dispersion=0
WQ Output cell volume=0
WQ Output cell surface area=0
WQ Output cell continuity=0
WQ Output cumulative cell continuity=0
WQ Output face conc=0
WQ Output face dconc_dx=0
WQ Output face courant=0
WQ Output face peclet=0
WQ Output face adv mass=0
WQ Output face disp mass=0
WQ Output cell mass=0
WQ Output cell source sink temp=0
WQ Output cell source sink nsm=0
WQ Output MaxMinRange=-1
WQ Daily Max Min Mean=-1
WQ Daily Range=0
WQ Daily Time=0
WQ Create Restart=0
WQ Fixed Restart=0
WQ System Summary=0
WQ Use Fixed Temperature=0
Sorting and Armoring Iterations= 10
XS Update Threshold= 0.02
Hydraulics Update Threshold= 0.02
Energy Slope Method= 1
Volume Change Method= 0
XS Weighting Method= 0
Number of US Weighted Cross Sections= 1
Number of DS Weighted Cross Sections= 1
Upstream XS Weight=0.25
Main XS Weight=0.5
Downstream XS Weight=0.25
Number of DS XS's Weighted with US Boundary= 1
Upstream Boundary Weight= 1
Weight of XSs Associated with US Boundary= 0
Number of US XS's Weighted with DS Boundary= 1
Downstream Boundary Weight= 0.5
Weight of XSs Associated with DS Boundary= 0.5
Sediment Output Level= 4
Mass or Volume Output= 0
Output Increment Type= 1
Profile and TS Output Increment= 10
XS Output Flag= 0
XS Output Increment= 10
Disregard all LS=0
Disregard all Conn=0
Disregard all Breaches=0
Disregard all Pumps=0

--- HOOSIER CREEK.f01 (steady flow) ---

Flow Title=Multiple
Program Version=4.10
Number of Profiles= 7
Profile Names=10-year,25-year,50-year,1pct_min,100-year,1pct_plu,500-year
River Rch & RM=HOOSIER CREEK,Reach-1         ,57725
     560     896    1197     775    1545    3084    2549
River Rch & RM=HOOSIER CREEK,Reach-1         ,57183
     680    1098    1476     959    1914    3820    3189
River Rch & RM=HOOSIER CREEK,Reach-1         ,54546
     941    1548    2106    1384    2762    5511    4707
River Rch & RM=HOOSIER CREEK,Reach-1         ,52097
     956    1573    2138    1405    2804    5594    4773
River Rch & RM=HOOSIER CREEK,Reach-1         ,49933
    1226    2038    2791    1845    3682    7346    6347
River Rch & RM=HOOSIER CREEK,Reach-1         ,45637
    1312    2188    3003    1989    3968    7917    6863
River Rch & RM=HOOSIER CREEK,Reach-1         ,44797
    1542    2590    3571    2374    4737    9453    8264
River Rch & RM=HOOSIER CREEK,Reach-1         ,40851
    1689    2846    3933    2619    5226   10427    9146
River Rch & RM=HOOSIER CREEK,Reach-1         ,37249
    2100    3570    4962    3323    6630   13228   11728
River Rch & RM=HOOSIER CREEK,Reach-1         ,34056
    2301    3927    5471    3672    7326   14618   13019
River Rch & RM=HOOSIER CREEK,Reach-1         ,32898
    2423    4142    5777    3881    7743   15449   13784
River Rch & RM=HOOSIER CREEK,Reach-1         ,30574
    2583    4424    6180    4156    8292   16545   14796
River Rch & RM=HOOSIER CREEK,Reach-1         ,28519
    2763    4738    6623    4455    8890   17737   15875
River Rch & RM=HOOSIER CREEK,Reach-1         ,24363
    2762    4734    6616    4450    8878   17715   15847
River Rch & RM=HOOSIER CREEK,Reach-1         ,23909
    2951    5070    7096    4779    9536   19027   17068
River Rch & RM=HOOSIER CREEK,Reach-1         ,21206
    3125    5378    7535    5079   10134   20220   18168
River Rch & RM=HOOSIER CREEK,Reach-1         ,16092
    3275    5610    7839    5268   10512   20973   18723
River Rch & RM=HOOSIER CREEK,Reach-1         ,7806
    3524    6059    8486    5716   11405   22757   20409
River Rch & RM=HOOSIER CREEK,Reach-1         ,6672
    3605    6200    8686    5852   11676   23297   20899
River Rch & RM=HOOSIER CREEK,Reach-1         ,3307
    3671    6316    8850    5963   11897   23737   21299
Boundary for River Rch & Prof#=HOOSIER CREEK,Reach-1         , 1
Up Type= 0
Dn Type= 3
Dn Slope=0.00206
Boundary for River Rch & Prof#=HOOSIER CREEK,Reach-1         , 2
Up Type= 0
Dn Type= 3
Dn Slope=0.00206
Boundary for River Rch & Prof#=HOOSIER CREEK,Reach-1         , 3
Up Type= 0
Dn Type= 3
Dn Slope=0.00206
Boundary for River Rch & Prof#=HOOSIER CREEK,Reach-1         , 4
Up Type= 0
Dn Type= 3
Dn Slope=0.00206
Boundary for River Rch & Prof#=HOOSIER CREEK,Reach-1         , 5
Up Type= 0
Dn Type= 3
Dn Slope=0.00206
Boundary for River Rch & Prof#=HOOSIER CREEK,Reach-1         , 6
Up Type= 0
Dn Type= 3
Dn Slope=0.00206
Boundary for River Rch & Prof#=HOOSIER CREEK,Reach-1         , 7
Up Type= 0
Dn Type= 3
Dn Slope=0.00206
DSS Import GetInterval= 0
DSS Import GetPeak= 0
DSS Import FillOption= 0

--- HOOSIER CREEK.g01 (geometry) ---

Geom Title=Existing Conditions
Program Version=4.10

River Reach=HOOSIER CREEK   ,Reach-1
Reach XY= 30
        2447475.       13517075.      2448622.55     13518069.53
      2451185.28     13518974.01       2452873.5     13518671.54
        2453025.       13518225.        2454350.     13518975.41
      2455135.45     13518175.53      2456878.31       13518467.
      2457376.48     13517578.61        2459425.       13517525.
      2459578.53     13516326.45      2460211.27      13515788.2
      2464849.89     13513124.68      2467614.57     13513276.05
      2469575.09     13514017.72      2470018.88     13513676.82
      2470876.65     13514671.89      2471695.16     13514494.63
      2471821.68     13515366.96       2476064.5      13515173.8
      2476774.97     13514432.48      2478714.81     13515675.46
      2479316.84     13515381.05      2479626.73     13514228.31
      2482728.42     13514767.21      2483218.94     13513483.14
      2484364.38     13513724.41      2485159.78     13513175.51
      2486818.93     13514816.89        2488825.       13515525.

Type RM Length L Ch R = 1 ,57725   ,542,542,542
BEGIN DESCRIPTION:
HOOSIER CREEK 106.0
END DESCRIPTION:
XS GIS Cut Line= 3
      2447224.97     13517475.03        2447625.       13517125.
      2448025.02     13516524.97
#Sta/Elev= 30
  4473.6  323.07  4615.5  320.46    4700  319.62  4820.5  317.35  4920.2  316.24
  4962.9  315.31  4969.6   314.9  4981.8  312.95    4982  312.45  4985.5  312.45
  4985.8  312.95    4998  314.32  5008.2  313.97  5012.7  314.53  5063.7  315.43
  5077.3  315.19  5099.8   315.9    5235  317.18    5250  316.95  5286.1  317.54
  5293.6  318.09  5365.7  318.07  5449.2  319.56  5517.4  320.38  5532.5  321.16
  5538.5  320.72  5568.5   321.5  5610.6  321.75  5712.7  324.18  5726.3  324.09
#Mann= 5 ,-1 , 0
  4473.6     .05       0  4920.2     .07       0  4981.8     .05       0
  4985.8     .07       0  5449.2     .12       0
Bank Sta=4981.8,4985.8
XS Rating Curve= 0 ,0
Exp/Cntr=0.3,0.1

Type RM Length L Ch R = 1 ,57183   ,352,352,352
BEGIN DESCRIPTION:
Mapping XS 8a9b8dea
END DESCRIPTION:
XS GIS Cut Line= 3
      2447642.81     13517750.73      2447986.98     13517442.41
      2448237.34       13517049.
#Sta/Elev= 30
  4497.7  318.92  4517.3  318.52  4524.4  318.73  4545.7  318.03  4574.1  317.83
  4585.2  317.03  4673.6  315.72  4715.5  315.66  4743.8  314.86  4843.3   313.5
  4878.4  313.48  4942.7  312.67  4992.3  312.79  5013.7  311.71  5013.9  311.21
  5017.4  311.21  5017.7  311.71  5036.8  312.77  5051.5  313.12    5058  313.91
  5094.4  314.54    5152  314.71  5158.2  315.15  5188.4  315.09  5203.6  315.59
  5209.6  315.32    5250  316.28  5261.2  316.71  5282.4  316.55  5426.1  319.15
#Mann= 6 ,-1 , 0
  4497.7     .05       0  4524.4     .07       0  4585.2     .05       0
  5013.7     .05       0  5017.7     .05       0    5250     .12       0
Bank Sta=5013.7,5017.7
XS Rating Curve= 0 ,0
Exp/Cntr=0.3,0.1

Type RM Length L Ch R = 1 ,56831   ,462,462,462
BEGIN DESCRIPTION:
HOOSIER CREEK 104.0
END DESCRIPTION:
XS GIS Cut Line= 3
        2447875.       13518225.        2448225.       13517625.
      2448524.97     13517375.02
#Sta/Elev= 30
    4310  319.77  4339.4  319.38  4382.4  320.05  4398.1  319.16  4413.8  319.62
  4419.6  318.88  4484.1  318.93  4499.8  319.66  4506.8  318.73    4537  318.11
  4542.8  318.48  4564.7  317.37  4595.7  317.08  4601.5  316.34  4645.7  315.75
  4668.9  316.31  4697.4  314.79  4703.6  315.22  4981.5  310.72  4994.8  308.58
    4995  308.08  4998.5  308.08  4998.8  308.58  5001.7  310.74  5007.9  310.74
  5011.8  309.98  5018.3  311.24  5089.9  313.31  5210.9  314.79  5395.1  320.94
#Mann= 3 ,-1 , 0
    4310     .05       0  4994.8     .05       0  4998.8     .05       0
Bank Sta=4994.8,4998.8
XS Rating Curve= 0 ,0
Exp/Cntr=0.3,0.1

Type RM Length L Ch R = 1 ,56369   ,486,486,486
BEGIN DESCRIPTION:
HOOSIER CREEK 103.0
END DESCRIPTION:
XS GIS Cut Line= 3
        2448475.     13518524.97        2448475.       13517975.
      2448725.01     13517374.97
#Sta/Elev= 30
  4445.9  320.97  4495.9  320.11  4515.9  319.14    4578  317.79  4625.9  316.57
  4656.6  316.58  4705.9  315.45  4735.9  315.28  4775.9  313.93  4785.9  313.77
  4795.9  314.25  4885.9  311.62  4955.9  310.22  4975.9  309.29  4998.6  308.94
  5008.5  308.14  5008.7  307.64  5012.2  307.64  5012.5  308.14  5017.5  308.94
  5034.3  310.12  5071.7  309.63  5104.2   310.9    5180   311.7  5294.3  313.87
  5477.4  318.72  5515.9  320.18  5606.8  322.38  5613.4   322.9  5645.9  323.52
#Mann= 6 ,-1 , 0
  4445.9     .05       0    4578    .035       0  4656.6     .05       0
  5008.5     .05       0  5012.5     .05       0  5606.8     .07       0
Bank Sta=5008.5,5012.5
XS Rating Curve= 0 ,0
Exp/Cntr=0.3,0.1

Type RM Length L Ch R = 1 ,55883   ,457,457,457
BEGIN DESCRIPTION:
HOOSIER CREEK 102.0
END DESCRIPTION:
XS GIS Cut Line= 3
      2448674.97     13518375.03        2448925.       13518075.
        2448875.     13517525.02
#Sta/Elev= 30
  4609.1  316.11  4657.7   315.1  4786.8  312.02  4836.3  311.31  4857.1  310.45
  4885.8  310.13  4928.7  308.45  4935.2  308.52    4943  307.39  4949.5  307.95
  4967.6  305.64  4978.2  304.37  4990.5  303.49  4990.7  302.99  4994.2  302.99
  4994.5  303.49  5009.7  303.57  5019.7  304.27  5029.8   305.6  5059.9  312.08
  5069.9  312.32    5090  310.23  5110.1  309.81  5170.4   310.6  5200.5  311.59
  5220.6  311.53  5264.9  312.58  5275.8  312.51    5331  313.82  5551.9  320.63
#Mann= 6 ,-1 , 0
  4609.1    .035       0  4657.7     .05       0  4967.6     .07       0
  4990.5     .05       0  4994.5     .07       0  5264.9     .12       0
Bank Sta=4990.5,4994.5
XS Rating Curve= 0 ,0
Exp/Cntr=0.3,0.1

Type RM Length L Ch R = 1 ,55426   ,436,436,436
BEGIN DESCRIPTION:
HOOSIER CREEK 101.0
END DESCRIPTION:
XS GIS Cut Line= 3
      2448725.03     13518774.97        2449325.       13518175.
      2449924.99     13517575.01
#Sta/Elev= 30
  4156.3  322.96  4241.1  321.53  4538.1  313.51  4576.1  312.94  4594.7  313.07
  4622.9  312.14  4665.4  312.28  4679.5  311.07  4715.3  309.92  4820.9  307.83
  4962.4  307.09  4977.5  306.63  4988.6  306.55  4988.9  306.05  4992.4  306.05
  4992.6  306.55  5033.1  306.91  5061.4  306.62  5117.9  308.51  5132.1  308.47
  5177.1  309.48  5202.8  308.01  5217.6  310.41  5344.2  311.88  5488.7  314.87
  5624.3  317.74  5796.7   322.2  5810.9  323.03    5825  322.91  5853.3   323.6
#Mann= 10 ,-1 , 0
  4156.3     .05       0  4576.1    .035       0  4715.3     .05       0
  4977.5     .07       0  4988.6     .05       0  4992.6     .07       0
  5177.1    .035       0  5217.6     .07       0  5488.7     .12       0
  5624.3     .07       0
Bank Sta=4988.6,4992.6
XS Rating Curve= 0 ,0
Exp/Cntr=0.3,0.1

Type RM Length L Ch R = 1 ,54990   ,444,444,444
BEGIN DESCRIPTION:
HOOSIER CREEK 100.0
END DESCRIPTION:
XS GIS Cut Line= 3
      2449075.04     13518874.97        2449675.       13518325.
      2450125.01     13517724.99
#Sta/Elev= 30
  4181.7  318.03    4393  313.54  4658.6  307.97  4711.3  307.64  4803.9  306.24
  4852.7  306.17  4868.3  305.05  4889.2  307.98  4912.2  306.44  5021.7  304.47
    5022  303.97  5025.7  304.47  5273.7  309.22    5282  311.26  5338.3  310.95
  5395.6  313.98  5467.5  313.83    5482  314.78  5509.1  320.84  5545.5  320.92
  5588.3  316.41    5682  321.19  5688.3  324.04  5702.9  323.31  5709.1  326.83
  5717.5  324.54  5723.7  326.79    5732  325.29  5738.3  328.99  5745.6  326.91
#Mann= 10 ,-1 , 0
  4181.7     .07       0    4393    .035       0  4658.6     .05       0
  4711.3    .035       0  4803.9     .12       0  4852.7    .035       0
  4912.2     .12       0  5021.7     .05       0  5025.7     .12       0
  5545.5     .07       0
Bank Sta=5021.7,5025.7
XS Rating Curve= 0 ,0
Exp/Cntr=0.3,0.1

Type RM Length L Ch R = 1 ,54546   ,339,339,339
BEGIN DESCRIPTION:
HOOSIER CREEK 99.0
END DESCRIPTION:
XS GIS Cut Line= 3
      2449675.02     13519074.96        2449975.       13518475.
      2450324.99     13517825.02
#Sta/Elev= 30
  4321.8  315.86  4495.4  311.41  4576.1  309.11  4604.1  310.37  4644.2  309.05
  4940.1  303.44  4947.9  300.64  4961.8  300.27  4978.6  302.21  4984.2  300.84
  5000.7  302.94  5044.5  303.07    5070  299.17  5070.2  298.67  5074.2  299.17
  5082.6  301.77  5088.3  300.81  5094.8  303.48  5279.8  307.49    5356  312.47
  5383.6  312.09  5412.8  306.06  5495.7  307.63  5601.4  310.79  5628.6  312.38
  5640.8  316.78  5662.7  320.22    5717   323.6  5722.7  327.49  5730.8  325.97
#Mann= 9 ,-1 , 0
  4321.8     .05       0  4495.4     .07       0  4604.1    .035       0
  4644.2     .07       0  4940.1     .12       0    5070     .05       0
  5074.2     .12       0  5495.7     .07       0  5601.4     .12       0
Bank Sta=5070,5074.2
XS Rating Curve= 0 ,0
Exp/Cntr=0.3,0.1

Type RM Length L Ch R = 1 ,54207   ,237,237,237
BEGIN DESCRIPTION:
HOOSIER CREEK 98.0
END DESCRIPTION:
XS GIS Cut Line= 3
      2449905.46     13519186.83      2450255.13      13518554.7
      2450563.51      13517992.3
#Sta/Elev= 30
  4277.6   313.6  4302.2   313.5    4314  312.58  4345.8  313.13  4359.7  311.97
  4373.2  312.61  4433.2  311.87  4514.1  311.89  4530.1  310.33  4565.4  309.11
  4908.6  303.42  4921.5  303.25  4953.9  302.08  4976.8  298.75  5007.7  300.22
  5016.8  298.31  5020.4  297.52  5020.6  297.02  5024.6  297.52  5029.6  298.36
  5035.3  303.09  5136.7  303.88  5238.2  305.62  5301.6  306.56  5348.9  308.27
  5352.4  308.33  5459.6  311.49  5568.2  314.16  5570.3  314.19  5641.4  316.17
#Mann= 14 ,-1 , 0
  4277.6    .035       0  4433.2     .07       0  4908.6     .12       0
  4921.5    .035       0  5016.8     .12       0  5020.4    .035       0
  5024.6     .12       0  5136.7    .035       0  5238.2     .12       0
  5348.9     .07       0  5352.4     .12       0  5459.6     .07       0
  5568.2    .035       0  5570.3     .07       0
#XS Ineff= 2 ,-1
    4278    4839     310    5186    5641     310
Permanent Ineff=
       F       F
Bank Sta=5020.4,5024.6
XS Rating Curve= 0 ,0
Exp/Cntr=0.3,0.1

Type RM Length L Ch R = 1 ,53970   ,242,242,242
BEGIN DESCRIPTION:
HOOSIER CREEK 97.0
END DESCRIPTION:
XS GIS Cut Line= 3
      2450105.18     13519237.09        2450465.     13518625.02
      2450797.86     13518091.31
#Sta/Elev= 30
    4290  310.15  4597.7  306.66  4689.8  306.21    4753  305.32  4853.5  303.59
  4893.7  303.32  4933.6   302.5    4942  301.77  4949.2  300.58    4955  300.41
  4977.9  298.14    4990  298.11  4990.3  297.61    4994  297.61  4994.3  298.11
  4997.1  298.82  5013.6  299.16    5023  300.37  5028.9   300.3  5035.4  301.02
  5093.2  301.24  5205.9  302.79  5312.1  304.86  5348.9  305.95    5443  308.41
  5485.5  308.88  5537.4  310.19  5543.3  309.94  5595.2  311.51    5629  311.78
#Mann= 10 ,-1 , 0
    4290    .035       0  4689.8     .07       0    4753    .035       0
  4893.7     .07       0  4977.9    .063       0    4990     .05       0
  4994.3    .063       0  5093.2     .07       0  5205.9    .063       0
  5348.9     .07       0
#XS Ineff= 2 ,-1
    4290    4890     310    5190    5629     310
Permanent Ineff=
       F       F
Bank Sta=4990,4994.3
XS Rating Curve= 0 ,0
Exp/Cntr=0.3,0.1

Type RM Length L Ch R = 1 ,53728   ,514,514,514
BEGIN DESCRIPTION:
Mapping XS 2932d416
END DESCRIPTION:
XS GIS Cut Line= 3
      2450292.66     13519200.67      2450693.71     13518586.07
       2450922.9      13518190.2
#Sta/Elev= 30
  4271.1  306.44  4275.6  306.48  4522.5  303.85  4579.8  304.08    4595  305.16
  4798.2  301.92  4847.7  301.67  4926.8  301.28  4978.1  297.37  4993.3  297.29
    4997  295.47  4997.3  294.97  5001.4  295.47  5002.6  297.28  5008.5  297.28
  5014.8  299.76  5020.5  298.61  5057.8  302.37  5079.4  301.66  5087.1  302.76
  5116.7   303.3  5122.4  302.15  5132.4  303.42  5138.2  302.53  5153.9  304.04
  5181.3  303.63  5191.1   305.1  5214.5  305.55  5449.2  310.05  5462.4  310.46
#Mann= 8 ,-1 , 0
  4271.1    .035       0  4275.6     .05       0  4798.2     .07       0
  4847.7     .12       0    4997     .05       0  5001.4     .12       0
  5214.5     .07       0  5449.2    .035       0
Bank Sta=4997,5001.4
XS Rating Curve= 0 ,0
Exp/Cntr=0.3,0.1

Type RM Length L Ch R = 1 ,53214   ,430,430,430
BEGIN DESCRIPTION:
HOOSIER CREEK 96.0
END DESCRIPTION:
XS GIS Cut Line= 3
      2450875.01     13519274.96        2451025.       13518825.
      2451225.03     13518574.97
#Sta/Elev= 30
  4520.8  307.78    4700  302.71  4797.8  300.92  4879.2  298.78  4942.8  299.65
    4974  298.76  4992.5  296.89  4998.3  296.89  5002.3  294.45  5014.4  291.78
  5014.8  291.28  5018.7  291.28    5019  291.78  5031.1  295.35  5037.5  296.69
  5045.5  297.81  5051.9  297.78  5072.7  300.58  5087.1  300.27  5095.1  300.79
  5101.6  299.93  5109.6  301.08    5116  300.69  5123.2  301.65    5180  303.13
  5208.8  305.38  5251.2  305.96  5272.8   307.2  5293.6  307.65  5315.3  307.12
#Mann= 5 ,-1 , 0
  4520.8     .05       0  4797.8     .07       0  4942.8     .12       0
  5014.4     .05       0    5019     .12       0
Bank Sta=5014.4,5019
XS Rating Curve= 0 ,0
Exp/Cntr=0.3,0.1

Type RM Length L Ch R = 1 ,52784   ,220,220,220
BEGIN DESCRIPTION:
HOOSIER CREEK 95.0
END DESCRIPTION:
XS GIS Cut Line= 3
        2451275.       13519375.        2451375.       13518975.
        2451375.     13518625.01
#Sta/Elev= 30
  4587.7  305.84  4701.1  303.52  4711.4  302.82  4762.9  301.69  4770.7  301.11
  4775.8  301.35  4891.5   298.9  4907.2  298.83  4935.6  297.28  4940.7  297.78
  4969.1  295.01  4976.8  293.14    4982  293.42  4989.7  290.49  4995.1  289.77
  4995.4  289.27  4999.4  289.27  4999.8  289.77  5002.5  289.77    5010  293.08
    5020  294.75    5050   297.7    5080  298.05    5160  300.38    5170  300.21
    5240  302.33    5280  303.78    5290  304.64    5310  304.75    5350  306.98
#Mann= 4 ,-1 , 0
  4587.7     .05       0  4891.5     .12       0  4995.1     .05       0
  4999.8     .12       0
Bank Sta=4995.1,4999.8
XS Rating Curve= 0 ,0
Exp/Cntr=0.3,0.1

Type RM Length L Ch R = 1 ,52564   ,246,246,246
BEGIN DESCRIPTION:
Mapping XS f0e5a473
END DESCRIPTION:
XS GIS Cut Line= 3
      2451442.75     13519431.13      2451595.53     13519004.06
      2451578.18     13518639.75
#Sta/Elev= 30
  4517.7  306.32  4565.1  304.87  4587.9  304.72  4657.5  302.07  4688.2  301.79
  4694.1  301.38  4829.5   298.6  4853.4  298.19    4949  297.82  4954.6  296.26
  4990.4   297.1  5000.4   293.4    5008  289.48  5008.4  288.98  5012.4  288.98
  5012.7  289.48  5020.4  289.52  5030.4  292.23  5070.4  294.76  5086.5  296.57
  5091.5   296.5  5120.5  298.08  5130.5  298.13  5170.6  299.93  5210.6  301.18
  5230.6  303.06  5240.6  302.82  5270.7  303.49  5301.7  304.44    5336  306.12
#Mann= 4 ,-1 , 0
  4517.7     .05       0  4829.5     .12       0    5008     .05       0
  5012.7     .12       0
Bank Sta=5008,5012.7
XS Rating Curve= 0 ,0
Exp/Cntr=0.3,0.1

Type RM Length L Ch R = 1 ,52318   ,221,221,221
BEGIN DESCRIPTION:
HOOSIER CREEK 94.0
END DESCRIPTION:
XS GIS Cut Line= 3
      2451624.99     13519425.02        2451825.       13518925.
      2451724.99     13518624.97
#Sta/Elev= 30
  4457.6  305.33  4526.3  304.25    4534  303.05  4550.5  301.62  4640.7  299.66
  4651.5  299.94  4658.2  299.18  4780.7  297.97  4825.2  296.81  4849.4  294.72
  4856.1  293.08  4866.9  292.43  4873.6  293.37    4879  292.11  4903.2  290.76
  4920.7  294.12  4951.7  292.62  4957.1  293.41  4974.6  289.69  4984.2  289.01
  4984.5  288.51  4988.9  288.51  4989.3  289.01  4998.8   289.1  5017.2  292.26
  5038.3  292.32  5080.5   296.6    5091  296.33  5175.3  300.88  5312.4  305.62
#Mann= 4 ,-1 , 0
  4457.6     .05       0    4534     .12       0  4984.2     .05       0
  4989.3     .12       0
Bank Sta=4984.2,4989.3
XS Rating Curve= 0 ,0
Exp/Cntr=0.3,0.1

Type RM Length L Ch R = 1 ,52097   ,238,238,238
BEGIN DESCRIPTION:
Mapping XS 5099b60e
END DESCRIPTION:
XS GIS Cut Line= 3
      2452154.55     13519404.79      2452000.48     13518792.83
      2451823.09      13518559.2
#Sta/Elev= 30
  4347.5  299.52  4369.6   299.8  4543.2  297.84  4563.8  298.32  4645.1  297.18
  4718.5  297.35  4759.8  296.37  4821.7  296.18  4873.2  295.26  4898.8  295.95
  4904.1   294.8  4914.5  293.93  4934.7  292.87  4939.9  293.43    4966  290.98
  4978.6  291.18  4988.4  289.15    4999  287.85  4999.4  287.35  5003.8  287.35
  5004.1  287.85  5009.8  290.65  5024.4  293.89  5030.6   296.1  5138.8  301.96
  5188.7  303.62  5194.9  303.28  5239.2  304.34  5265.7   305.1  5271.9  304.67
#Mann= 5 ,-1 , 0
  4347.5     .07       0  4645.1     .12       0    4999     .05       0
  5004.1     .12       0  5239.2     .07       0
Bank Sta=4999,5004.1
XS Rating Curve= 0 ,0
Exp/Cntr=0.3,0.1

Type RM Length L Ch R = 1 ,51859   ,437,437,437
BEGIN DESCRIPTION:
HOOSIER CREEK 93.0
END DESCRIPTION:
XS GIS Cut Line= 3
      2452475.01     13519475.02        2452225.       13518775.
      2451911.51     13518324.09
#Sta/Elev= 30
  4256.8  302.72  4359.3  300.77  4390.1  300.98  4395.4  302.02  4408.4  301.22
  4446.4  299.41  4681.5  297.49    4749  297.05  4798.4  294.51  4805.3   295.9
  4851.5  294.94  4861.6  293.93  4866.9  291.59  4872.7  291.44  4923.1  291.28
  4928.4     293  4953.9  292.21  4959.2  293.18  4968.3  291.43  4976.3  287.36
  4976.7  286.86  4981.5  287.36    4990  287.89  4997.5  290.23  5022.4  290.29
  5058.2  293.94  5222.3  296.33  5293.8  298.61  5368.4  299.26  5549.3  304.12
#Mann= 7 ,-1 , 0
  4256.8     .12       0  4408.4     .07       0  4681.5     .12       0
  4976.3     .05       0  4981.5     .12       0  5222.3     .07       0
  5368.4    .035       0
Bank Sta=4976.3,4981.5
XS Rating Curve= 0 ,0
Exp/Cntr=0.3,0.1

Type RM Length L Ch R = 1 ,51422   ,765,765,765
BEGIN DESCRIPTION:
HOOSIER CREEK 92.0
END DESCRIPTION:
XS GIS Cut Line= 3
      2452786.94     13519242.84        2452475.       13518475.
      2451984.42     13518180.65
#Sta/Elev= 30
  4177.8  298.92    4218  298.54  4223.4  299.17  4240.2  298.37  4461.7  297.45
  4574.8  297.66  4723.5  295.79  4866.3  291.96    4931  291.54  4962.4  290.55
  4974.2  288.85    4985  288.31  5011.7  287.77  5012.2  287.27    5017  287.77
  5115.4  292.03  5122.4  291.58  5158.2  291.49  5183.6  290.33  5195.1  290.06
  5204.8  291.26  5280.8  292.52  5321.5  293.14  5333.1  294.57  5348.7  295.05
    5370   295.1    5407   297.5  5414.8  298.63  5473.1  299.87  5578.7  303.58
#Mann= 7 ,-1 , 0
  4177.8     .12       0  4723.5     .07       0  5011.7     .05       0
    5017     .07       0  5122.4    .035       0  5183.6     .07       0
  5280.8    .035       0
Bank Sta=5011.7,5017
XS Rating Curve= 0 ,0
Exp/Cntr=0.3,0.1

Type RM Length L Ch R = 1 ,50657   ,724,724,724
BEGIN DESCRIPTION:
Mapping XS 70a3a28c
END DESCRIPTION:
XS GIS Cut Line= 4
      2452959.67     13519097.39      2453020.44     13518656.83
      2452751.34     13518331.31      2452417.33     13517891.31
#Sta/Elev= 30
  4465.1  296.57  4482.8  296.19  4936.8  291.74  4969.3  282.93  4969.7  282.43
  4974.6  282.93  5007.1  288.03  5078.8   287.5  5177.8  291.72  5255.9  290.44
  5270.3  287.49  5276.7   290.5  5284.6  286.48  5291.1  289.36  5298.9  286.71
  5305.4  290.29  5313.3   288.6  5326.5  291.86  5340.4   291.6  5348.7  288.17
  5354.9  289.88  5363.2  286.66  5419.4   290.5  5427.7  287.58    5463  291.57
  5483.9  291.83  5504.7  288.45  5527.9  290.57  5750.7  295.98  5884.6  297.79
#Mann= 6 ,-1 , 0
  4465.1     .12       0  4482.8     .07       0  4969.3     .05       0
  4974.6     .07       0  5527.9     .12       0  5750.7     .07       0
Bank Sta=4969.3,4974.6
XS Rating Curve= 0 ,0
Exp/Cntr=0.3,0.1

Type RM Length L Ch R = 1 ,49933   ,358,358,358
BEGIN DESCRIPTION:
HOOSIER CREEK 90.0
END DESCRIPTION:
XS GIS Cut Line= 3
      2453036.19     13519057.85      2453295.18     13518224.57
      2453302.54     13517868.94
#Sta/Elev= 30
  4127.4  295.61  4151.7  295.04  4183.6  295.09  4350.3  292.39  4533.4  291.31
  4622.6  290.31    4633  288.39  4647.2  287.12    4654  286.95  4664.4  288.78
  4674.5   286.8  4685.4  286.09  4695.9  289.61  4723.3  290.04  4815.2  289.75
  4842.5  290.32  4880.3  289.66  4926.2  285.82  4989.1   284.7  4997.2  282.73
  5002.3  282.73  5009.6  281.25  5026.5  280.42    5027  279.92  5032.6  280.42
  5069.6  286.95  5079.6  289.83  5089.6  294.01  5149.6  295.16  5355.7   302.4
#Mann= 7 ,-1 , 0
  4127.4     .07       0  4151.7     .12       0  4183.6     .07       0
  4533.4     .12       0  4723.3     .07       0  5026.5     .05       0
  5032.6     .07       0
Bank Sta=5026.5,5032.6
XS Rating Curve= 0 ,0
Exp/Cntr=0.3,0.1

Type RM Length L Ch R = 1 ,49575   ,418,418,418
BEGIN DESCRIPTION:
HOOSIER CREEK 89.0
END DESCRIPTION:
XS GIS Cut Line= 3
      2453175.01     13519074.99        2453525.       13518475.
      2453574.99     13518175.05
#Sta/Elev= 30
  4311.4  297.33  4322.9  296.95  4405.2  293.07    4494  291.71  4531.4  290.55
  4575.6  285.67  4602.9  285.68  4612.4   289.7  4618.6  290.13  4683.1  288.43
    4693  289.74  4698.8  288.28  4728.2  290.07  4751.3  287.92  4773.2  289.53
    4786  286.58  4794.7  287.35  4800.5   282.8  4912.2  283.55  4917.9  284.78
  4933.7  282.97  5008.5   282.7  5030.8  278.83  5031.3  278.33    5037  278.83
    5039  281.84  5046.6  283.75  5107.4  283.83  5155.5  291.62  5310.1  294.68
#Mann= 5 ,-1 , 0
  4311.4     .07       0  4322.9     .12       0    4494     .07       0
  5030.8     .05       0    5037     .07       0
Bank Sta=5030.8,5037
XS Rating Curve= 0 ,0
Exp/Cntr=0.3,0.1

Type RM Length L Ch R = 1 ,49157   ,417,417,417
BEGIN DESCRIPTION:
HOOSIER CREEK 88.0
END DESCRIPTION:
XS GIS Cut Line= 3
      2453724.99     13519075.05        2453775.       13518775.
        2453775.     13518224.99
#Sta/Elev= 30
  4700.6  293.97  4742.6   292.8  4812.2  290.18  4871.2  288.85  4890.8  288.45
    4911  287.18  4933.8  283.36  4954.1  281.37  4971.8  281.55  4984.5  278.75
  4991.4  278.08  4991.9  277.58  4997.4  277.58  4997.9  278.08  5002.3   280.1
  5024.8  280.38  5034.8  282.23  5044.8  282.98  5054.8  286.41  5074.8  288.17
  5104.8  287.28  5114.8  286.52  5124.8  284.98  5154.8  284.63  5184.8  285.72
  5224.8  288.16  5401.9  290.55  5414.8  291.38  5444.8  291.16  5554.8  294.08
#Mann= 7 ,-1 , 0
  4700.6     .12       0  4742.6     .07       0  4871.2     .12       0
  4890.8     .07       0  4991.4     .05       0  4997.9     .07       0
  5401.9     .12       0
Bank Sta=4991.4,4997.9
XS Rating Curve= 0 ,0
Exp/Cntr=0.3,0.1

Type RM Length L Ch R = 1 ,48740   ,930,930,930
BEGIN DESCRIPTION:
HOOSIER CREEK 87.0
END DESCRIPTION:
XS GIS Cut Line= 3
      2453990.06     13519081.37      2454095.09     13518644.21
        2453925.       13518275.
#Sta/Elev= 30
  4550.4  293.67  4742.1  286.84  4760.8  285.34    4766  283.84  4772.9  283.17
  4783.2  284.01  4793.5  286.73  4811.5  286.79  4865.5   284.4  4886.1  284.17
  4916.9  281.64    4939  281.73    4958  278.38  5010.6  276.34  5011.1  275.84
  5017.2  276.34  5021.1  280.93  5059.8  280.23  5076.2  281.27  5082.8  282.62
  5088.3  282.14  5105.7  283.58  5111.2  283.04  5128.7   284.6  5134.2  283.49
  5151.7  285.22  5157.2  284.67  5174.6  287.54  5294.9  289.07  5406.5  292.05
#Mann= 4 ,-1 , 0
  4550.4     .12       0  4811.5     .07       0  5010.6     .05       0
  5017.2     .07       0
Bank Sta=5010.6,5017.2
XS Rating Curve= 0 ,0
Exp/Cntr=0.3,0.1

Type RM Length L Ch R = 1 ,47810   ,467,467,467
BEGIN DESCRIPTION:
HOOSIER CREEK 86.0
END DESCRIPTION:
XS GIS Cut Line= 3
        2454675.     13519025.05        2454675.       13518775.
      2454025.01     13517975.02
#Sta/Elev= 30
  4754.7  290.07  4894.7  284.91  4924.7  283.13  4945.6  279.61  4954.7   278.5
  4964.7  274.12  4971.4  273.38  4971.9  272.88    4978  273.38  4994.7  275.74
  5002.2   277.9    5008   277.9  5018.4  280.07  5026.3  280.12  5032.7  283.06
  5040.7  281.06    5055   281.2  5061.5  282.28  5075.9   279.4  5096.7  283.46
  5133.3   285.1  5345.9  285.09  5381.1  283.54  5417.1   285.5  5601.7  287.25
  5737.4  290.06  5798.4  292.13  5829.8   292.7  5913.9  295.63  6035.5  299.45
#Mann= 7 ,-1 , 0
  4754.7     .12       0  4945.6     .07       0  4971.4     .05       0
    4978     .07       0  5798.4     .12       0  5829.8     .07       0
  5913.9     .12       0
Bank Sta=4971.4,4978
XS Rating Curve= 0 ,0
Exp/Cntr=0.3,0.1

Type RM Length L Ch R = 1 ,47343   ,884,884,884
BEGIN DESCRIPTION:
HOOSIER CREEK 85.0
END DESCRIPTION:
XS GIS Cut Line= 3
        2455075.     13518874.99        2455075.       13518575.
      2454725.02     13517925.03
#Sta/Elev= 30
  4695.8  288.97  4955.8   284.4  4965.8  281.92  4985.8  279.74  4993.3  275.21
  4998.6  275.21  5000.6  273.21  5001.1  272.71  5007.3  273.21  5018.5  274.26
  5031.5  277.11  5085.8  278.68  5107.7  278.09  5129.7   280.1  5135.3  281.88
  5195.4  280.03    5201  281.41  5239.2  282.87  5268.4   282.8  5277.3  282.33
  5291.1  277.36  5304.9  275.45  5321.1  276.73  5326.8  278.83  5336.5  278.89
  5348.7  281.45  5370.6  283.35  5381.1  281.93  5386.8  283.37    5734  291.01
#Mann= 3 ,-1 , 0
  4695.8     .07       0  5000.6     .05       0  5007.3     .07       0
Bank Sta=5000.6,5007.3
XS Rating Curve= 0 ,0
Exp/Cntr=0.3,0.1

Type RM Length L Ch R = 1 ,46459   ,473,473,473
BEGIN DESCRIPTION:
HOOSIER CREEK 84.0
END DESCRIPTION:
XS GIS Cut Line= 3
      2455174.98     13518775.02        2455525.       13518275.
        2455525.     13517924.96
#Sta/Elev= 30
  4394.1  286.84  4717.2  281.23  4723.7  279.36    4732   279.9  4760.3  275.42
  4767.7  278.81  4773.8  276.89  4782.6  280.07  4788.7  278.75  4803.5     279
  4809.6  276.33  4833.1  275.53  4904.6  276.16  4910.7  275.52  4925.6  276.96
  4940.4  276.77  4946.5  275.84  4955.2  276.41  4990.9  274.76    4997  273.59
  5044.5  273.67  5060.9  271.83  5061.4  271.33    5068  271.83  5094.5  274.15
  5114.5  274.61  5154.5  278.99  5194.5  279.93  5264.5  284.59  5354.5     287
#Mann= 3 ,-1 , 0
  4394.1     .07       0  5060.9     .05       0    5068     .07       0
Bank Sta=5060.9,5068
XS Rating Curve= 0 ,0
Exp/Cntr=0.3,0.1

Type RM Length L Ch R = 1 ,45986   ,349,349,349
BEGIN DESCRIPTION:
HOOSIER CREEK 83.0
END DESCRIPTION:
XS GIS Cut Line= 3
      2455374.99     13518925.01        2455725.       13518525.
      2455925.01     13518074.97
#Sta/Elev= 30
  4464.5  286.25  4581.9   284.8    4689  283.62  4773.9  283.25  4825.7  283.22
  4861.7  282.11    4876  282.85  4889.7  281.56  4960.4  280.23    4968  276.41
  4988.9  273.86  4992.7  272.43  5014.4  270.78  5014.9  270.28  5021.5  270.78
  5028.2  272.92  5062.4  274.61  5072.6  277.58  5085.6  277.58  5103.4  275.76
  5122.7   276.4  5132.1  276.67  5155.4  279.49  5201.9     279  5207.4  278.13
  5230.6  278.76  5259.3  277.15  5304.5  280.51  5433.8  285.94  5488.5  286.68
#Mann= 8 ,-1 , 0
  4464.5     .12       0  4581.9     .07       0    4689     .12       0
  4773.9     .07       0  5014.4     .05       0  5021.5     .07       0
  5122.7     .12       0  5304.5     .07       0
Bank Sta=5014.4,5021.5
XS Rating Curve= 0 ,0
Exp/Cntr=0.3,0.1

Type RM Length L Ch R = 1 ,45637   ,267,267,267
BEGIN DESCRIPTION:
HOOSIER CREEK 82.0
END DESCRIPTION:
XS GIS Cut Line= 3
      2455974.44     13519055.33      2456014.86     13518374.43
      2456052.43     13518129.09
#Sta/Elev= 30
  4317.9   284.3  4416.4  283.48  4429.1  283.64  4488.5  282.75  4498.5   283.5
  4518.6  282.65  4538.6  282.91  4558.7  282.22  4627.1  281.54  4698.9  281.22
  4739.3  280.36    4779  280.15  4809.1  278.85  4859.2  278.41  4916.1  274.18
  4979.4   270.6  4985.6  268.88  4986.1  268.38  4992.8  268.38  4993.3  268.88
  5002.2  269.01  5009.5  271.64  5034.4  274.43  5039.9  275.49  5097.8  280.61
  5102.8  280.05  5110.7  280.89  5161.1  282.87  5225.6  284.14  5248.2  284.87
#Mann= 8 ,-1 , 0
  4317.9     .07       0  4416.4     .12       0  4429.1     .07       0
  4627.1     .12       0  4739.3     .07       0  4985.6     .05       0
  4993.3     .07       0  5225.6     .12       0
Bank Sta=4985.6,4993.3
XS Rating Curve= 0 ,0
Exp/Cntr=0.3,0.1

Type RM Length L Ch R = 1 ,45370   ,573,573,573
BEGIN DESCRIPTION:
Mapping XS 818b2ff7
END DESCRIPTION:
XS GIS Cut Line= 4
      2456019.01     13519089.27      2456117.98     13518667.36
      2456269.02     13518401.74      2456289.81     13517939.13
#Sta/Elev= 30
  4383.9  285.08  4480.8  283.17  4735.5  281.48  4777.9  280.23  4788.9  278.49
  4819.3  278.57  4823.5  276.96  4839.4  279.64  4866.8     280  4876.9  279.65
    4889  277.67  4898.5  278.13  4904.3  276.46    4935  272.33  4947.5  272.55
  4957.6  271.09  4979.2  271.42  4992.5  269.91    4997  267.05  4997.5  266.55
  5004.7  267.05  5006.6  270.94  5081.6  275.74  5087.3   274.8  5129.6   273.3
  5144.6  275.75  5149.6  274.68  5189.6  277.63  5249.7  279.76  5585.9  285.34
#Mann= 3 ,-1 , 0
  4383.9     .07       0    4997     .05       0  5004.7     .07       0
Bank Sta=4997,5004.7
XS Rating Curve= 0 ,0
Exp/Cntr=0.3,0.1

Type RM Length L Ch R = 1 ,44797   ,569,569,569
BEGIN DESCRIPTION:
Mapping XS 75dfa547
END DESCRIPTION:
XS GIS Cut Line= 4
      2456659.74     13519017.48      2456588.55     13518577.92
      2456531.05     13518226.58      2456418.85     13517938.88
#Sta/Elev= 30
  4198.7  287.01  4282.2  286.87  4318.4  285.54  4448.3   282.2  4525.4  279.11
  4578.9  278.87  4638.4  278.71  4694.7  276.61  4738.1  275.92  4756.1  273.69
  4798.9  271.54  4849.6  271.28  4859.7  270.63  4869.9  270.83  4883.9  272.32
  4961.1  271.29  4991.5  269.26  4998.3  267.66  5008.5  266.74    5009  266.24
  5015.8  266.24  5016.3  266.74  5029.5  272.33  5034.8  272.05    5054  276.86
  5059.3  275.99  5098.3  279.23  5246.9  282.16  5291.5  284.39  5308.8  284.02
#Mann= 5 ,-1 , 0
  4198.7     .07       0  4318.4     .12       0  4578.9     .07       0
  5008.5     .05       0  5016.3     .07       0
Bank Sta=5008.5,5016.3
XS Rating Curve= 0 ,0
Exp/Cntr=0.3,0.1

Type RM Length L Ch R = 1 ,44228   ,295,295,295
BEGIN DESCRIPTION:
Mapping XS 9502d692
END DESCRIPTION:
XS GIS Cut Line= 3
      2457260.33     13518837.49      2456973.88     13518386.11
      2456522.49     13517743.75
#Sta/Elev= 30
  4494.2   284.5  4730.4  281.25  4849.3  280.03  4917.3  278.26  4935.4  277.82
    4942  272.11  4947.9  274.71  4957.3  272.59  4963.2  276.74  4970.9  276.02
  4978.4   271.1  4984.4  271.25  4993.7  267.09  4995.5  263.38    4996  262.88
  5003.8  263.38  5006.4   265.9  5020.8  269.25  5056.8  271.02    5079  270.61
  5122.2   275.8    5137   276.4  5345.2  276.53  5553.5  279.09  5580.5  280.46
    5604  278.95    5631   279.8  5681.6  278.24  5696.4     276  5813.9  281.73
#Mann= 6 ,-1 , 0
  4494.2     .05       0  4730.4     .07       0  4849.3     .12       0
  4917.3     .07       0  4995.5     .05       0  5003.8     .07       0
Bank Sta=4995.5,5003.8
XS Rating Curve= 0 ,0
Exp/Cntr=0.3,0.1

Type RM Length L Ch R = 1 ,43933   ,545,545,545
BEGIN DESCRIPTION:
Mapping XS 3ecf0339
END DESCRIPTION:
XS GIS Cut Line= 3
      2457624.89     13518768.02      2457199.57      13518212.5
      2456722.14      13517630.9
#Sta/Elev= 30
  4328.8  285.15  4611.4  280.99  4887.4  278.65  4950.8  277.78  4965.3  276.01
  4972.9  270.35  4987.5  268.15  4996.5  263.52    4997  263.02  5004.8  263.52
  5023.4  268.21  5051.1  268.21  5113.7   273.1  5179.7  275.11    5207  273.45
  5229.2  273.57  5264.4  268.73  5278.7  273.32  5307.5  274.42  5363.4  275.14
  5377.8  276.39  5385.6  278.56    5400  279.21  5420.8  272.91  5569.3  272.87
  5591.6  275.94    5598  275.74  5605.9  277.73  5633.3   279.5  5780.9  281.79
#Mann= 8 ,-1 , 0
  4328.8     .05       0  4611.4     .07       0  4887.4     .12       0
  4972.9     .07       0  4996.5     .05       0  5004.8     .07       0
  5113.7     .12       0  5307.5     .07       0
Bank Sta=4996.5,5004.8
XS Rating Curve= 0 ,0
Exp/Cntr=0.3,0.1

Type RM Length L Ch R = 1 ,43388   ,431,431,431
BEGIN DESCRIPTION:
Mapping XS 696277d9
END DESCRIPTION:
XS GIS Cut Line= 3
      2457885.34     13518637.86      2457407.91     13517830.56
      2456730.85     13517535.43
#Sta/Elev= 30
    3917  284.32  3952.7  283.91  4391.8  277.78  4745.2  275.29  4923.5  272.49
  4935.6  271.67  4953.6  268.01  4967.2  267.26    4989  263.29  4999.9  262.12
  5005.9  263.07    5007  261.77  5007.5  261.27  5015.8  261.77  5021.7  266.06
  5029.3  265.75  5034.8  264.36  5052.7   267.6  5133.9  268.68  5151.9  269.88
  5163.5  272.23  5180.8  273.92  5218.1  276.35  5233.1  278.54  5279.9  278.77
  5316.3  280.63  5384.5  282.22  5436.8  282.96  5501.6  282.31  5593.5  283.86
#Mann= 5 ,-1 , 0
    3917     .07       0  3952.7     .05       0  4391.8     .07       0
    5007     .05       0  5015.8     .07       0
Bank Sta=5007,5015.8
XS Rating Curve= 0 ,0
Exp/Cntr=0.3,0.1

Type RM Length L Ch R = 1 ,42957   ,431,431,431
BEGIN DESCRIPTION:
Mapping XS 79cd8efa
END DESCRIPTION:
XS GIS Cut Line= 3
      2457954.77      13518507.6       2457590.2      13517587.5
      2457321.12      13517110.1
#Sta/Elev= 30
  3938.2  282.44  3978.5  281.96  4002.8  280.96  4016.3  281.23  4344.1  276.78
  4494.5  275.29  4518.8  274.46    4608  274.12    4780  275.59  4794.4  275.12
  4801.5  273.25  4818.7  270.76    4866  271.46  4897.1   266.4  4919.8  266.98
  4954.1  265.54    4970  263.88  4976.7  260.81  4981.3  260.51  4981.8  260.01
    4990  260.01  4990.5  260.51  4999.6  266.94  5007.6  271.33  5013.3  272.46
  5045.2   273.5  5088.5  276.35    5122  277.52  5333.6  285.78  5475.9  290.06
#Mann= 6 ,-1 , 0
  3938.2     .05       0  4344.1     .07       0  4981.3     .05       0
  4990.5     .07       0    5122    .035       0  5333.6     .07       0
Bank Sta=4981.3,4990.5
XS Rating Curve= 0 ,0
Exp/Cntr=0.3,0.1

Type RM Length L Ch R = 1 ,42526   ,595,595,595
BEGIN DESCRIPTION:
Mapping XS 04a83c6a
END DESCRIPTION:
XS GIS Cut Line= 3
       2458215.2     13518412.15      2457972.14     13517561.46
      2457624.92     13517040.62
#Sta/Elev= 30
  4091.3  281.55  4296.9  278.64  4323.1  277.62  4552.1  274.64  4689.5  272.56
  4835.1  272.53  4879.3  273.75  4889.1  272.67  4941.1  271.56  4946.9  267.27
  4952.1  268.32  4961.9  263.89    4976  263.34  4978.8  261.21  4989.2  260.15
  4989.7  259.65  4998.6  260.15  5007.8  261.66  5014.9  265.33  5043.9  265.57
    5057  264.11  5123.1  265.92  5152.1  269.16  5159.1  268.96  5165.1  270.79
  5174.1  271.04  5180.1  272.14  5216.2  274.25  5404.4  279.89    5602  287.64
#Mann= 5 ,-1 , 0
  4091.3     .07       0  4323.1     .05       0  4552.1     .07       0
  4989.2     .05       0  4998.6     .07       0
Bank Sta=4989.2,4998.6
XS Rating Curve= 0 ,0
Exp/Cntr=0.3,0.1

Type RM Length L Ch R = 1 ,41931   ,542,542,542
BEGIN DESCRIPTION:
Mapping XS eeb92918
END DESCRIPTION:
XS GIS Cut Line= 3
      2458675.27     13518290.61      2458536.38     13517613.54
      2458015.85     13517049.63
#Sta/Elev= 30
  4256.7  283.51  4507.4  278.29  4640.1  272.22  4742.2  269.42  4823.9  267.39
  4861.3  268.02  4930.5  270.05  4936.2  267.53  4969.2  262.09    4976  263.11
  4983.3  258.39  4990.1  259.82  4997.5  257.44  5011.7  259.02  5025.9  258.62
    5028  257.34  5028.5  256.84  5037.4  257.34    5040  261.09  5046.8  259.42
  5054.2   262.6    5061  261.95  5075.2  266.92    5082   266.2  5089.4  268.34
  5103.5  269.13  5266.3  272.55  5449.6   274.4  5506.7   274.4  5715.3   281.3
#Mann= 5 ,-1 , 0
  4256.7     .05       0  4861.3     .07       0    5028     .05       0
  5037.4     .07       0  5449.6    .035       0
Bank Sta=5028,5037.4
XS Rating Curve= 0 ,0
Exp/Cntr=0.3,0.1

Type RM Length L Ch R = 1 ,41389   ,538,538,538
BEGIN DESCRIPTION:
Mapping XS 90bfda31
END DESCRIPTION:
XS GIS Cut Line= 3
       2459239.5     13518186.44      2459031.17     13517596.18
      2458406.16     13516953.81
#Sta/Elev= 30
    4344  285.02  4377.6   284.7  4419.8  282.45  4459.8  281.27  4552.6  280.32
    4600  278.77  4676.3  277.62  4758.5  274.85  4851.3  269.21  4938.7  266.08
    4950  264.59  4975.1  263.11  4982.3   261.6  4998.6  256.47  4999.1  255.97
  5007.7  255.97  5008.2  256.47  5010.6  257.83  5024.7  261.23  5074.1  261.92
  5109.6   265.6  5144.9  266.77    5152   268.5    5159  268.91  5203.8  269.28
  5238.1  269.62  5484.4  271.11  5562.1  272.66  5724.8  273.64  5866.2  276.23
#Mann= 5 ,-1 , 0
    4344     .07       0  4998.6     .05       0  5008.2     .07       0
  5203.8    .035       0  5238.1     .07       0
Bank Sta=4998.6,5008.2
XS Rating Curve= 0 ,0
Exp/Cntr=0.3,0.1

Type RM Length L Ch R = 1 ,40851   ,621,621,621
BEGIN DESCRIPTION:
Mapping XS dd795f4b
END DESCRIPTION:
XS GIS Cut Line= 3
      2459986.03     13517813.19      2459499.92     13517448.61
      2458719.35     13516919.56
#Sta/Elev= 30
    4394  283.33  4415.9  282.79    4697   275.4  4800.4  273.14  4871.3  269.31
  4944.2  266.89  4950.4  265.84  4957.8  263.52    4965  259.82  4985.8  258.12
  5002.5  254.38    5003  253.88  5012.2  253.88  5012.7  254.38  5015.3  257.04
  5051.2  261.38  5102.1  263.56  5129.2  263.95  5152.5  262.97  5165.1  263.64
    5174  265.11  5201.1  265.58    5231  267.44  5317.8  267.01  5404.7  268.72
  5489.4  268.12  5597.6  268.77    5709  270.16    5781  270.82  5944.6  272.83
#Mann= 9 ,-1 , 0
    4394    .035       0  4415.9     .05       0    4697     .07       0
  5002.5     .05       0  5012.7     .07       0  5489.4    .035       0
  5597.6     .07       0    5709    .035       0    5781     .07       0
Bank Sta=5002.5,5012.7
XS Rating Curve= 0 ,0
Exp/Cntr=0.3,0.1

Type RM Length L Ch R = 1 ,40230   ,666,666,666
BEGIN DESCRIPTION:
Mapping XS b937d869
END DESCRIPTION:
XS GIS Cut Line= 3
      2460472.16     13517639.59      2459525.96     13516893.06
      2458719.33     13516624.18
#Sta/Elev= 30
  3817.1  285.18  3818.8   284.9    3839  281.91    3847  285.63  3941.3  285.71
  4159.6  283.92  4349.3  278.48  4394.1  276.86  4637.4  270.83    4900  267.06
  4921.7  266.04  4929.2  263.32    4950  259.44  4972.5  257.92  4978.9   255.8
  4980.3  252.17  4980.8  251.67  4990.5  252.17  4993.4  254.25  5007.8  255.18
  5019.8  258.19  5025.5  258.19  5030.3  261.32  5035.6  261.19    5055  263.88
  5067.2  263.76  5086.6  266.33  5188.5  265.45  5367.2  267.61  5872.6  275.93
#Mann= 10 ,-1 , 0
  3817.1     .07       0  3818.8    .035       0  3941.3     .05       0
  4349.3    .035       0  4394.1     .05       0    4900     .07       0
  4980.3     .05       0  4990.5     .07       0  5188.5    .035       0
  5367.2     .07       0
Bank Sta=4980.3,4990.5
XS Rating Curve= 0 ,0
Exp/Cntr=0.3,0.1

Type RM Length L Ch R = 1 ,39564   ,445,445,445
BEGIN DESCRIPTION:
Mapping XS cdfb512b
END DESCRIPTION:
XS GIS Cut Line= 3
      2460671.77     13517422.54      2459795.06     13516372.22
      2458935.68     13516016.32
#Sta/Elev= 30
  3426.7  286.45  3557.3  282.99  3576.2  284.38  3606.8  281.88    3707  280.27
  3735.6  274.71  3742.1  276.88  3756.4  275.55  3762.9  278.12  3777.2  278.81
  4017.4  274.17  4037.7   273.6  4214.5  270.09  4444.9  266.37    4743  265.11
  4859.8  257.91  4901.5  258.99  4960.1  256.89  4984.4  252.11  4984.9  251.61
    4995  252.11  5066.5  258.01  5085.2  262.09    5098  265.79  5114.2  264.08
  5119.6  265.82  5173.7  268.59  5371.5  272.32    5721  277.92    5725  277.94
#Mann= 10 ,-1 , 0
  3426.7     .07       0  3576.2     .12       0  4017.4     .07       0
  4037.7     .12       0  4214.5     .07       0  4984.4     .05       0
    4995     .07       0  5085.2     .12       0  5371.5    .035       0
    5721     .07       0
Bank Sta=4984.4,4995
XS Rating Curve= 0 ,0
Exp/Cntr=0.3,0.1

Type RM Length L Ch R = 1 ,39119   ,359,359,359
BEGIN DESCRIPTION:
Mapping XS 746f7c65
END DESCRIPTION:
XS GIS Cut Line= 3
      2460888.78     13517231.56      2460038.12     13516146.53
       2459318.8     13515704.54
#Sta/Elev= 30
  3559.9   285.2  3688.3  284.01  3841.3  279.51  3880.8  280.22  4168.6  271.35
  4179.2  268.65  4216.2  265.59  4251.5  266.31  4257.8  269.26  4272.3  269.69
  4286.7  266.45  4301.2   266.1    4322   269.4  4349.2   268.5  4411.3  267.46
  4461.5  266.67  4763.2  263.22  4905.3  264.05  4955.5  262.54  4965.1  257.47
  4965.6  250.81  4966.1  250.31  4976.3  250.81  5013.5  255.19    5081  257.42
  5130.1  263.83  5160.3  262.32    5197  265.65  5300.7   268.3  5782.9  279.67
#Mann= 11 ,-1 , 0
  3559.9     .07       0  3841.3     .12       0  4168.6     .07       0
  4349.2     .12       0  4411.3    .035       0  4461.5     .07       0
  4763.2     .12       0  4905.3     .07       0  4965.6     .05       0
  4976.3     .07       0  5300.7    .035       0
Bank Sta=4965.6,4976.3
XS Rating Curve= 0 ,0
Exp/Cntr=0.3,0.1

Type RM Length L Ch R = 1 ,38760   ,664,664,664
BEGIN DESCRIPTION:
Mapping XS ae9df6e4
END DESCRIPTION:
XS GIS Cut Line= 3
      2461244.73     13516893.08      2460203.05     13515842.71
      2459700.03     13515634.56
#Sta/Elev= 30
  3492.3   278.4    3816  276.03  4032.7  271.02  4266.2  267.23  4516.1  263.15
  4544.4  264.05  4650.4  262.48  4678.7  260.72  4699.9  255.58    4707  255.37
  4714.1  257.71  4721.1  257.98  4728.2  261.57  4742.4   262.2  4777.7  261.52
  4798.9  259.04  4862.5  260.03  4897.9  257.32  4954.4  256.38  4982.2  251.99
  4985.8  249.12  4986.3  248.62  4996.5  249.12  5000.7  252.61    5030  253.62
  5045.3  256.46  5053.9  261.67  5066.9  265.94  5272.5  271.94    5516  277.07
#Mann= 5 ,-1 , 0
  3492.3     .07       0  4032.7    .035       0  4266.2     .07       0
  4985.8     .05       0  4996.5     .12       0
Bank Sta=4985.8,4996.5
XS Rating Curve= 0 ,0
Exp/Cntr=0.3,0.1

Type RM Length L Ch R = 1 ,38096   ,328,328,328
BEGIN DESCRIPTION:
Mapping XS 2b7f97e4
END DESCRIPTION:
XS GIS Cut Line= 3
      2461765.53     13516754.16       2460758.6     13515825.35
      2459865.17     13515469.71
#Sta/Elev= 30
  3605.3     274  3654.7  273.55  3661.5  271.74  3697.2  274.04  3798.4  272.61
  3824.2  271.33  3909.3  272.35  4083.3  271.01  4200.3  270.08  4772.9  264.74
  4921.9  261.67  4942.5  260.73    4964  252.51  4974.2  249.91  4979.8  249.91
  4981.5  245.43    4982  244.93  4992.5  245.43  5000.6  251.12  5016.7  253.43
  5110.7  258.74  5120.7  259.06  5235.1  261.25    5302     262  5310.7  256.18
  5323.5  258.38  5334.2   262.6  5340.4  263.09  5506.1  266.18  5936.8  279.48
#Mann= 11 ,-1 , 0
  3605.3     .07       0  3798.4     .12       0  4083.3     .07       0
  4200.3     .12       0  4921.9     .07       0  4981.5     .05       0
  4992.5     .07       0  5110.7      .1       0  5120.7     .12       0
  5235.1     .07       0  5506.1     .12       0
Bank Sta=4981.5,4992.5
XS Rating Curve= 0 ,0
Exp/Cntr=0.3,0.1
