--- JOHNS CREEK.prj (project) ---

Proj Title=JOHNS CREEK Base Level Engineering
Current Plan=p01
Default Exp/Contr=0.3,0.1
English Units
Geom File=g01
Flow File=f01
Plan File=p01
Y Axis Title=Elevation
X Axis Title(PF)=Main Channel Distance
X Axis Title(XS)=Station
BEGIN DESCRIPTION:
JOHNS CREEK
END DESCRIPTION:
DSS Export Rating Curves= 0
DSS Export Rating Curve Sorted= 0
DSS Export Volume Flow Curves= 0
DXF OffsetX= 0
DXF OffsetY= 0
DXF ScaleX= 1
DXF ScaleY= 10

--- JOHNS CREEK.p01 (plan) ---

Plan Title=Multiple Run
Program Version=4.10
Short Identifier=Multiple
Geom File=g01
Flow File=f01
Subcritical Flow
K Sum by GR= 0
Std Step Tol= 0.01
Critical Tol= 0.01
Num of Std Step Trials= 20
Max Error Tol= 0.3
Flow Tol Ratio= 0.001
Split Flow NTrial= 30
Split Flow Tol= 0.02
Split Flow Ratio= 0.02
Log Output Level= 0
Friction Slope Method= 1
Unsteady Friction Slope Method= 2
Unsteady Bridges Friction Slope Method= 1
Parabolic Critical Depth
Global Vel Dist= 1 , 1 , 1
Global Log Level= 0
CheckData=True
Encroach Param=-1 ,0,0, 0
BEGIN DESCRIPTION:
Multiple Run
END DESCRIPTION:
Computation Interval=1HOUR
Output Interval=1HOUR
Run HTab= 0
Run UNet= 0
Run PostProcess= 0
Run WQNet= 0
UNET Theta= 1
UNET Theta Warmup= 1
UNET ZTol= 0.02
UNET ZSATol= 0.05
UNET MxIter= 20
UNET MaxInSteps= 0
UNET DtIC= 0
UNET DtMin= 0
UNET MaxCRTS= 20
UNET WFStab= 2
UNET SFStab= 1
UNET WFX= 1
UNET SFX= 1
UNET DSS MLevel= 4
UNET DZMax Abort= 100
UNET Convert EG Bridges= 0
UNET Use Existing IB Tables=-1
UNET Froude Reduction=False
UNET Froude Limit= 1
UNET Froude Power= 10
UNET Time Slicing=0,0, 5
UNET Junction Losses=0
Instantaneous Interval=1HOUR
Write IC File= 0
Write IC File at Sim End=0
Echo Input=False
Echo Parameters=False
Echo Output=False
Write Detailed= 0
WQ AD Non Conservative
WQ ULTIMATE=-1
WQ Max Comp Step=1HOUR
WQ Output Interval=15MIN
WQ Output Selected Increments= 0
WQ Output face flow=0
WQ Output face velocity=0
WQ Output face area=0
WQ Output face dispersion=0
WQ Output cell volume=0
WQ Output cell surface area=0
WQ Output cell continuity=0
WQ Output cumulative cell continuity=0
WQ Output face conc=0
WQ Output face dconc_dx=0
WQ Output face courant=0
WQ Output face peclet=0
WQ Output face adv mass=0
WQ Output face disp mass=0
WQ Output cell mass=0
WQ Output cell source sink temp=0
WQ Output cell source sink nsm=0
WQ Output MaxMinRange=-1
WQ Daily Max Min Mean=-1
WQ Daily Range=0
WQ Daily Time=0
WQ Create Restart=0
WQ Fixed Restart=0
WQ System Summary=0
WQ Use Fixed Temperature=0
Sorting and Armoring Iterations= 10
XS Update Threshold= 0.02
Hydraulics Update Threshold= 0.02
Energy Slope Method= 1
Volume Change Method= 0
XS Weighting Method= 0
Number of US Weighted Cross Sections= 1
Number of DS Weighted Cross Sections= 1
Upstream XS Weight=0.25
Main XS Weight=0.5
Downstream XS Weight=0.25
Number of DS XS's Weighted with US Boundary= 1
Upstream Boundary Weight= 1
Weight of XSs Associated with US Boundary= 0
Number of US XS's Weighted with DS Boundary= 1
Downstream Boundary Weight= 0.5
Weight of XSs Associated with DS Boundary= 0.5
Sediment Output Level= 4
Mass or Volume Output= 0
Output Increment Type= 1
Profile and TS Output Increment= 10
XS Output Flag= 0
XS Output Increment= 10
Disregard all LS=0
Disregard all Conn=0
Disregard all Breaches=0
Disregard all Pumps=0

--- JOHNS CREEK.f01 (steady flow) ---

Flow Title=Multiple
Number of Profiles=7
Profile Names=10-year,25-year,50-year,1pct_min,100-year,1pct_plu,500-year
River Rch & RM= JOHNS CREEK,Reach-1,19885
     687    1102    1474     954    1904    3800    3143
River Rch & RM= JOHNS CREEK,Reach-1,19433
     896    1456    1965    1282    2557    5102    4285
River Rch & RM= JOHNS CREEK,Reach-1,16635
    1055    1727    2343    1535    3063    6112    5180
River Rch & RM= JOHNS CREEK,Reach-1,14409
    1231    2027    2759    1813    3617    7217    6154
River Rch & RM= JOHNS CREEK,Reach-1,9318
    1293    2132    2905    1910    3810    7603    6490
River Rch & RM= JOHNS CREEK,Reach-1,6369
    1417    2345    3202    2109    4209    8397    7195
Boundary for River Rch & Prof#=JOHNS CREEK,Reach-1,1
Up Type=0
Dn Type=3
Dn Slope=0.005
Boundary for River Rch & Prof#=JOHNS CREEK,Reach-1,2
Up Type=0
Dn Type=3
Dn Slope=0.005
Boundary for River Rch & Prof#=JOHNS CREEK,Reach-1,3
Up Type=0
Dn Type=3
Dn Slope=0.005
Boundary for River Rch & Prof#=JOHNS CREEK,Reach-1,4
Up Type=0
Dn Type=3
Dn Slope=0.005
Boundary for River Rch & Prof#=JOHNS CREEK,Reach-1,5
Up Type=0
Dn Type=3
Dn Slope=0.005
Boundary for River Rch & Prof#=JOHNS CREEK,Reach-1,6
Up Type=0
Dn Type=3
Dn Slope=0.005
Boundary for River Rch & Prof#=JOHNS CREEK,Reach-1,7
Up Type=0
Dn Type=3
Dn Slope=0.005

--- JOHNS CREEK.g01 (geometry) ---

Geom Title=Existing Conditions
Program Version=4.10

River Reach=JOHNS CREEK     ,Reach-1
Reach XY= 30
        2520525.       13511575.      2521570.24     13511269.42
      2521651.48     13510897.87        2522217.     13510631.33
      2522024.52     13510395.17      2522251.64     13510147.44
      2522535.11      13510214.7      2522807.34     13509691.41
      2524422.56     13508530.47      2525223.41     13508671.18
      2525769.94     13508277.29      2525629.59     13508030.26
      2526085.64     13507825.55      2526723.53     13508171.47
      2526967.92       13507875.      2526811.66     13507488.33
      2527823.44     13507421.24      2527837.93     13507111.37
      2528281.05     13506876.58      2528514.25     13507124.32
      2529255.11     13506674.89      2529522.45     13507070.02
      2529823.75     13506971.49      2529625.53     13506585.68
      2530008.21     13505791.39      2530521.42     13506167.51
       2531073.5     13506071.53      2531422.94     13505669.15
      2531388.46     13505061.43        2531975.       13504975.

Type RM Length L Ch R = 1 ,19885   ,452,452,452
BEGIN DESCRIPTION:
JOHNS CREEK 36.0
END DESCRIPTION:
XS GIS Cut Line= 3
      2520374.98     13512325.04        2520775.       13511525.
        2520675.       13511225.
#Sta/Elev= 30
  4105.5  195.16  4127.9  195.22  4401.7  188.48  4537.7  186.13  4588.9  185.53
  4790.3  183.45  4829.5  181.68  4843.5  182.25  4851.8  179.41  4855.4  177.03
  4855.7  176.53  4859.4  177.03  4865.8   180.4  4874.2  180.35  4879.8  179.34
  4896.6  180.18  4902.1  178.13  4918.9  180.16  4924.5  178.05  4941.3  179.77
  4946.9  178.49  4955.3  180.43  4963.6  180.76    4986  180.26  4991.6  179.09
  5031.6  183.09  5131.2  184.73  5168.6  185.78  5263.6  189.45  5316.2  192.04
#Mann= 9 ,-1 , 0
  4105.5     .05       0  4401.7     .12       0  4537.7    .035       0
  4588.9     .12       0  4855.4     .05       0  4859.4     .12       0
  5131.2      .1       0  5168.6     .07       0  5263.6     .12       0
Bank Sta=4855.4,4859.4
XS Rating Curve= 0 ,0
Exp/Cntr=0.3,0.1

Type RM Length L Ch R = 1 ,19433   ,457,457,457
BEGIN DESCRIPTION:
JOHNS CREEK 35.0
END DESCRIPTION:
XS GIS Cut Line= 3
      2521325.01     13512225.02        2521125.       13511425.
        2520925.       13511125.
#Sta/Elev= 30
  4175.1  197.67  4247.3   197.2  4267.9  195.01  4275.6  193.54  4320.6  192.34
  4336.2  192.04  4494.7  187.96  4587.4  186.46  4693.1  183.84  4736.2  183.74
  4775.6  182.09    4858  181.46  4938.2     180  4976.6  178.88  4997.2  175.74
  5002.7  175.74  5005.2  174.66  5005.4  174.16  5009.1  174.16  5009.4  174.66
  5013.3  174.66  5028.3  178.81  5043.3  180.21  5107.9  181.26  5168.7  183.62
  5190.1  184.48  5208.6  185.02  5223.6  186.39  5280.7   189.3  5360.3  192.48
#Mann= 9 ,-1 , 0
  4175.1    .035       0  4320.6     .07       0  4336.2     .05       0
  4736.2     .07       0  4938.2      .1       0  5005.2     .05       0
  5009.4      .1       0  5168.7     .12       0  5190.1     .07       0
Bank Sta=5005.2,5009.4
XS Rating Curve= 0 ,0
Exp/Cntr=0.3,0.1

Type RM Length L Ch R = 1 ,18976   ,445,445,445
BEGIN DESCRIPTION:
JOHNS CREEK 34.0
END DESCRIPTION:
XS GIS Cut Line= 3
      2521974.98     13511974.96        2521525.       13511275.
      2521125.02     13510925.02
#Sta/Elev= 30
  4172.9  195.96  4681.9  183.78    4738  182.79  4767.3  181.46  4773.5  182.14
  4779.5  181.05  4788.7  181.78  4794.7     181  4802.9  182.31  4829.2  181.78
  4882.5  175.72  4888.5  176.21  4895.5  173.96  4895.8  173.46  4899.8  173.96
  4909.9  175.11  4918.8  177.48  4924.8  177.68  4991.5  177.15  5012.1  178.04
  5047.3  177.65  5075.7  178.77  5167.8  179.08  5281.7  182.33  5359.5  185.68
    5388  185.86  5416.5  187.79  5437.3  187.78  5503.8  190.63  5536.5  191.89
#Mann= 7 ,-1 , 0
  4172.9     .05       0  4681.9     .12       0    4738     .07       0
  4829.2     .12       0  4895.5     .05       0  4899.8     .12       0
  5503.8     .07       0
Bank Sta=4895.5,4899.8
XS Rating Curve= 0 ,0
Exp/Cntr=0.3,0.1

Type RM Length L Ch R = 1 ,18531   ,416,416,416
BEGIN DESCRIPTION:
JOHNS CREEK 33.0
END DESCRIPTION:
XS GIS Cut Line= 3
      2521824.99     13511674.97        2521625.       13510925.
      2521325.01       13510875.
#Sta/Elev= 30
  4223.5  187.77  4254.5  187.47  4409.8  183.89  4441.5  183.65  4504.6  182.27
    4534   181.7  4544.3  182.09  4585.7  180.89  4637.4  180.43  4647.8  180.71
  4666.6  179.88  4697.3  179.26  4714.7  178.96  4798.7  178.33  4821.8  178.07
  4861.9  178.37  4925.2   177.4  4947.9  176.11    4977   175.3  4989.3  173.69
  5007.7   172.9  5007.9   172.4  5011.7   172.4    5012   172.9    5020  173.33
  5032.6  174.96  5050.4  179.69  5182.2   184.6  5279.2  186.96  5303.8  187.51
#Mann= 9 ,-1 , 0
  4223.5     .05       0  4504.6     .07       0  4697.3     .12       0
  4714.7     .07       0  4798.7     .12       0  4925.2     .07       0
  5007.7     .05       0    5012     .07       0  5279.2     .12       0
Bank Sta=5007.7,5012
XS Rating Curve= 0 ,0
Exp/Cntr=0.3,0.1

Type RM Length L Ch R = 1 ,18115   ,376,376,376
BEGIN DESCRIPTION:
JOHNS CREEK 32.0
END DESCRIPTION:
XS GIS Cut Line= 3
      2522775.01     13511275.01        2521975.       13510825.
      2521524.97     13510574.99
#Sta/Elev= 30
  4082.6  194.95  4177.3  192.47  4243.2  189.86  4398.4  185.18  4472.7  183.78
    4553  180.57    4576  180.73    4615  179.02  4700.6  177.19  4792.4  176.59
  4846.6  176.45  4897.2   174.9  4954.9  174.92  4965.1  172.56  4986.8  175.33
  4992.5  173.95  5003.3  174.11  5008.5  170.61  5011.8  169.08  5012.2  168.58
  5016.3  168.58  5016.6  169.08  5023.4  169.86    5036  174.06    5068  174.85
  5089.7     176  5095.2  176.87  5149.2  177.44  5286.5   181.1  5515.3  185.04
#Mann= 6 ,-1 , 0
  4082.6     .05       0    4615     .12       0  4792.4      .1       0
  5011.8     .05       0  5016.6      .1       0  5095.2     .12       0
Bank Sta=5011.8,5016.6
XS Rating Curve= 0 ,0
Exp/Cntr=0.3,0.1

Type RM Length L Ch R = 1 ,17739   ,627,627,627
BEGIN DESCRIPTION:
JOHNS CREEK 31.0
END DESCRIPTION:
XS GIS Cut Line= 3
      2522674.99     13510924.99      2522226.18     13510590.41
      2521549.45     13510463.13
#Sta/Elev= 30
  4440.2  185.42  4739.5  177.08  4873.9  174.65  4976.5   174.4  4983.4  168.51
  4987.2   168.1  4987.5   167.6  4991.6   167.6    4992   168.1  4997.6  170.68
  5004.3  171.28  5011.4  173.26  5021.6  173.77  5082.6  174.04  5114.3  173.39
  5153.8  174.49  5174.2  171.98  5184.4  172.04  5235.2  176.11  5298.5  179.46
  5387.9  184.21  5439.4  185.92  5539.3  186.45  5544.4  187.08  5596.9  186.96
    5602  187.75  5632.1  187.18  5649.4  187.25  5654.5  187.95  5688.6  187.47
#Mann= 5 ,-1 , 0
  4440.2     .05       0  4873.9      .1       0  4987.2     .05       0
    4992      .1       0  5298.5     .12       0
Bank Sta=4987.2,4992
XS Rating Curve= 0 ,0
Exp/Cntr=0.3,0.1

Type RM Length L Ch R = 1 ,17112   ,477,477,477
BEGIN DESCRIPTION:
Mapping XS 5e7343bd
END DESCRIPTION:
XS GIS Cut Line= 3
       2522772.9     13510775.54      2522152.22     13510241.67
      2521758.65     13510077.33
#Sta/Elev= 30
  4185.6  184.08  4560.4  174.54  4574.7  174.68  4609.8  173.57  4638.1  173.84
  4687.7  173.36    4816  174.45  4908.3  173.67  4943.4  172.27  4971.9  170.16
  4986.2  170.46  4996.8  169.01  4997.1  168.51  5001.2  168.51  5001.6  169.01
  5007.7  169.07    5023  174.55  5027.5   174.8  5031.5  175.03  5032.4   175.7
  5036.9  179.02  5060.7  180.22  5084.5  180.43  5089.9   181.5  5161.4  183.94
  5174.7  185.18  5214.4  185.73  5254.6   187.7  5338.8  191.22  5430.8  195.24
#Mann= 8 ,-1 , 0
  4185.6     .05       0  4638.1      .1       0  4996.8     .05       0
  5001.6      .1       0  5027.5     .12       0  5032.4     .05       0
  5254.6     .12       0  5338.8     .05       0
Bank Sta=4996.8,5001.6
XS Rating Curve= 0 ,0
Exp/Cntr=0.3,0.1

Type RM Length L Ch R = 1 ,16635   ,321,321,321
BEGIN DESCRIPTION:
Mapping XS 40d153e7
END DESCRIPTION:
XS GIS Cut Line= 3
      2522959.52     13510610.61      2522403.96     13510055.04
       2521922.2     13509890.11
#Sta/Elev= 30
  4420.9  184.35  4442.9  183.43  4604.8  178.98  4838.2  174.87  4906.6  172.99
  4947.6  171.27  4972.5  169.97  4991.3  166.37  4991.6  165.87  4995.8  165.87
  4996.2  166.37  5000.8  168.18  5007.9  169.44    5015  169.91  5036.2  169.38
  5043.2  170.21  5064.5  171.14  5128.1  171.71  5156.4  173.21  5208.1  174.24
  5216.8  174.59  5353.5  183.49  5440.8  186.41  5459.2  187.58  5472.1  187.49
  5522.6  189.56  5554.3  189.81    5660  192.33  5670.6  193.06  5715.8  193.65
#Mann= 8 ,-1 , 0
  4420.9     .12       0  4442.9     .05       0  4906.6      .1       0
  4947.6     .05       0  4991.3     .05       0  4996.2     .05       0
  5208.1     .12       0  5216.8     .05       0
Bank Sta=4991.3,4996.2
XS Rating Curve= 0 ,0
Exp/Cntr=0.3,0.1

Type RM Length L Ch R = 1 ,16314   ,544,544,544
BEGIN DESCRIPTION:
Mapping XS 1bc41679
END DESCRIPTION:
XS GIS Cut Line= 3
      2523320.35     13510598.02      2522599.85      13509929.6
      2521923.83     13509669.59
#Sta/Elev= 30
  3996.1  193.23  4079.9  190.75    4098  189.41  4299.4  182.97  4447.9  178.26
  4582.2  175.78  4610.6  176.16  4674.1  172.78  4787.5  170.97  4865.1  172.11
  4900.8  169.94  4938.7  169.18  4946.1  168.68  4971.7  168.45  4978.5  167.32
  5005.8  166.07  5006.2  165.57  5010.8  166.07    5027  171.84  5032.9  172.62
  5080.5  173.94  5123.4   176.5  5166.2  176.76  5172.2  177.98  5181.3  177.42
  5219.8  178.29  5226.8  179.85  5241.2  181.08  5450.8  187.35  5703.2  192.41
#Mann= 8 ,-1 , 0
  3996.1     .12       0    4098     .05       0  4299.4     .12       0
  4938.7     .05       0  4946.1     .12       0  5005.8     .05       0
  5010.8     .12       0  5181.3     .05       0
Bank Sta=5005.8,5010.8
XS Rating Curve= 0 ,0
Exp/Cntr=0.3,0.1

Type RM Length L Ch R = 1 ,15770   ,347,347,347
BEGIN DESCRIPTION:
Mapping XS f71167f6
END DESCRIPTION:
XS GIS Cut Line= 3
      2523293.72       13510233.      2522842.33     13509668.76
      2522431.18     13509218.65
#Sta/Elev= 30
  4285.2  183.27  4488.6  175.99  4716.5  170.05  4752.7  169.42  4887.2  170.54
    4916  170.18  4930.4  168.17  4965.6  167.82  4973.6  167.17    4980  167.78
    4987  166.48  4991.8  162.48  4992.2  161.98  4996.7  161.98  4997.1  162.48
  5015.4  163.35  5022.8  166.79  5029.6  166.62    5037  169.49  5043.8  169.07
  5051.2  170.62    5058  170.12  5075.7   170.9  5291.7  175.89  5311.3  175.86
  5440.4  178.02  5518.1  178.58  5539.7  179.51  5574.8  179.35  5617.4  180.87
#Mann= 6 ,-1 , 0
  4285.2     .05       0  4716.5      .1       0  4991.8     .05       0
  4997.1      .1       0  5075.7     .12       0  5311.3     .05       0
Bank Sta=4991.8,4997.1
XS Rating Curve= 0 ,0
Exp/Cntr=0.3,0.1

Type RM Length L Ch R = 1 ,15423   ,240,240,240
BEGIN DESCRIPTION:
JOHNS CREEK 27.0
END DESCRIPTION:
XS GIS Cut Line= 3
      2523324.98     13510024.95        2523175.       13509625.
      2522825.02     13509325.02
#Sta/Elev= 30
  4568.9   180.9  4614.2  179.11  4664.1  175.93  4749.5  172.39  4754.9  172.53
  4761.1  171.89  4789.1  171.25  4925.7  167.75  4986.3  167.87  4993.4   164.6
  4999.3   164.6  5003.2  162.78  5007.1  162.23  5007.5  161.73    5012  161.73
  5012.4  162.23    5024  164.59  5052.6  166.67  5081.1  167.04  5107.1  166.13
  5123.9  166.24  5144.8  167.38    5159  167.47  5180.4  168.46  5187.6  169.54
  5194.2  169.19  5208.4  170.56  5239.6  171.94  5322.6  175.57    5457  179.85
#Mann= 6 ,-1 , 0
  4568.9     .05       0  4789.1     .12       0  5007.1     .05       0
  5012.4     .12       0  5107.1      .1       0  5239.6     .05       0
Bank Sta=5007.1,5012.4
XS Rating Curve= 0 ,0
Exp/Cntr=0.3,0.1

Type RM Length L Ch R = 1 ,15183   ,233,233,233
BEGIN DESCRIPTION:
Mapping XS 10da5cf6
END DESCRIPTION:
XS GIS Cut Line= 3
      2523493.38     13509920.51      2523258.99     13509417.02
      2522899.37     13509226.38
#Sta/Elev= 30
  4424.9  180.39  4474.9  178.34  4491.5  177.04  4503.3  176.11  4585.9   172.9
  4595.9  172.61  4696.1  169.44  4737.6  168.16  4834.7  167.57  4872.2  166.26
    4936  167.61  4971.5  166.35  4977.4  164.51  4980.3  164.31  5007.7  163.78
  5014.8  162.87  5017.9  160.95  5018.3  160.45  5022.8  160.45  5023.2  160.95
  5036.8  161.53  5042.5  163.58  5058.8  164.97    5074  168.21  5086.7  169.12
  5141.1  170.34  5212.8     173  5222.5  173.96  5267.5  175.24  5387.3  180.75
#Mann= 10 ,-1 , 0
  4424.9     .05       0  4491.5     .12       0  4585.9     .07       0
  4595.9     .12       0  4696.1      .1       0    4936     .12       0
  5007.7      .1       0  5017.9     .05       0  5023.2      .1       0
    5074     .05       0
Bank Sta=5017.9,5023.2
XS Rating Curve= 0 ,0
Exp/Cntr=0.3,0.1

Type RM Length L Ch R = 1 ,14950   ,193,193,193
BEGIN DESCRIPTION:
JOHNS CREEK 26.0
END DESCRIPTION:
XS GIS Cut Line= 3
      2523675.02     13509675.03        2523425.       13509275.
      2523075.03     13509175.01
#Sta/Elev= 30
  4532.7   175.2  4650.1     170  4759.9  166.85  4790.8  166.06  4815.8  165.61
  4838.7  165.97  4851.1  166.64  4910.1  167.63  4945.5  167.41  4960.2  166.65
  4969.1  165.25  4981.4  164.48  4994.1  159.21  4994.5  158.71    4999  158.71
  4999.4  159.21  5001.5  160.59    5007  160.59  5014.8  161.58  5021.3  163.79
  5026.5  166.13  5060.3  167.33  5087.6   167.4  5127.6  168.15  5160.4  169.08
  5181.2  170.11  5295.6  172.73  5326.8  173.81  5346.3  175.17  5368.4  175.73
#Mann= 6 ,-1 , 0
  4532.7     .05       0  4759.9     .07       0  4790.8      .1       0
  4994.1     .05       0  4999.4      .1       0  5127.6     .05       0
Bank Sta=4994.1,4999.4
XS Rating Curve= 0 ,0
Exp/Cntr=0.3,0.1

Type RM Length L Ch R = 1 ,14757   ,348,348,348
BEGIN DESCRIPTION:
Mapping XS b67cf8f9
END DESCRIPTION:
XS GIS Cut Line= 3
      2523814.58     13509616.71       2523571.5     13509154.86
      2523169.38     13508981.53
#Sta/Elev= 30
  4503.2  173.59  4535.8  171.98  4648.9  168.63    4687   167.4  4726.6  166.99
  4754.3  165.58  4787.1  164.94  4889.3  167.37  4919.3  166.78  4941.3  167.08
  4957.2  166.28    4969  166.67  4979.7  166.04  4985.4  161.73  4991.1  159.41
  4999.1  159.25  4999.5  158.75    5004  158.75  5004.4  159.25  5007.4  161.21
  5013.7  163.94  5022.2   164.8  5108.1   165.1  5160.6  166.75    5166   166.1
  5173.8  167.08  5206.4  168.55  5312.6  169.97  5350.4  171.24    5463  174.92
#Mann= 7 ,-1 , 0
  4503.2     .05       0  4535.8     .07       0  4648.9     .12       0
    4687      .1       0  4999.1     .05       0  5004.4      .1       0
  5350.4     .05       0
Bank Sta=4999.1,5004.4
XS Rating Curve= 0 ,0
Exp/Cntr=0.3,0.1

Type RM Length L Ch R = 1 ,14409   ,324,324,324
BEGIN DESCRIPTION:
Mapping XS ae40e367
END DESCRIPTION:
XS GIS Cut Line= 4
      2523949.97     13509488.19      2523842.33     13508981.25
      2523772.89     13508884.03      2523342.83     13508599.64
#Sta/Elev= 30
  4428.9   171.1  4460.2  170.66  4670.9  167.21  4765.1  165.28  4786.6  164.06
  4814.7  162.35  4871.7  163.01  4908.9  164.89  4979.4  164.69  4985.6  163.01
  4991.7  163.27  5000.3  161.21  5006.4  162.18  5025.7  158.14  5026.2  157.64
  5031.4  158.14  5035.9  161.54  5042.1  161.67  5062.9  165.83    5078  166.88
  5100.1  167.19  5123.2  165.56  5159.3  167.66  5216.5     169  5237.5  170.41
  5252.6  170.04  5317.9  173.09  5439.1  175.62  5523.3  174.75  5582.2  173.85
#Mann= 7 ,-1 , 0
  4428.9      .1       0  4460.2     .12       0  4786.6      .1       0
  5025.7     .05       0  5031.4      .1       0  5317.9     .12       0
  5523.3      .1       0
Bank Sta=5025.7,5031.4
XS Rating Curve= 0 ,0
Exp/Cntr=0.3,0.1

Type RM Length L Ch R = 1 ,14085   ,260,260,260
BEGIN DESCRIPTION:
JOHNS CREEK 24.0
END DESCRIPTION:
XS GIS Cut Line= 3
      2524374.98     13509374.97        2524075.       13508975.
      2523674.97     13508574.97
#Sta/Elev= 30
  4500.3  175.01  4585.4  172.37  4593.4  172.05  4755.4  167.01  4762.7  166.84
  4928.4  165.53    4943  164.54  4957.6  162.09  4963.8  155.82  4969.2  155.48
  4969.7  154.98  4974.6  154.98  4975.1  155.48  4986.7  156.53  4997.1  159.09
  5003.8  159.09  5014.4  161.94    5071  163.36  5099.3  163.01  5127.5  165.02
  5155.8  165.85  5244.9  166.78  5339.7   167.1    5368  167.79  5382.1  166.61
  5410.4  169.06  5424.5  168.85  5463.3  173.39  5531.8   176.7    5566  178.21
#Mann= 10 ,-1 , 0
  4500.3     .12       0  4585.4     .07       0  4593.4      .1       0
  4755.4     .12       0  4762.7      .1       0  4969.2     .05       0
  4975.1      .1       0  5244.9    .063       0  5463.3     .12       0
  5531.8     .07       0
Bank Sta=4969.2,4975.1
XS Rating Curve= 0 ,0
Exp/Cntr=0.3,0.1

Type RM Length L Ch R = 1 ,13825   ,383,383,383
BEGIN DESCRIPTION:
Mapping XS 0551bbb4
END DESCRIPTION:
XS GIS Cut Line= 3
      2524608.83     13509269.47      2524257.26     13508796.36
      2523845.28     13508479.79
#Sta/Elev= 30
  4444.3  175.37  4528.5  172.72  4637.4  168.08  4793.5  163.79    4879  163.62
  4899.8   164.8  4914.4  163.22  4922.8  159.47  4964.5  161.56  4972.9  159.51
  4976.2  156.76  4976.7  156.26  4982.1  156.76  4999.9  159.03  5008.3  158.86
  5031.5  160.73  5053.5  161.05  5143.2  161.39  5172.2  164.03  5193.1  164.52
  5207.6  165.95    5251  166.18  5278.2  165.09  5342.6  166.35  5392.4  169.54
    5465  171.96  5500.3  174.85  5514.8  174.67  5521.5  175.59  5553.3  176.74
#Mann= 6 ,-1 , 0
  4444.3     .07       0  4637.4      .1       0  4976.2     .05       0
  4982.1      .1       0  5053.5    .035       0  5521.5     .12       0
Bank Sta=4976.2,4982.1
XS Rating Curve= 0 ,0
Exp/Cntr=0.3,0.1

Type RM Length L Ch R = 1 ,13442   ,342,342,342
BEGIN DESCRIPTION:
Mapping XS 5c1b1104
END DESCRIPTION:
XS GIS Cut Line= 3
      2524699.98     13509195.69      2524370.11     13508561.99
      2523979.74     13508323.43
#Sta/Elev= 30
  4298.8   174.8    4385  172.34  4454.5  169.61  4511.7  166.96  4644.3   163.1
    4852  163.13  4909.6  162.38    4926  161.13  4953.8  160.98  4964.6  159.42
  4970.2  157.09    4973  154.72  4973.5  154.22  4978.9  154.72  4992.4  156.81
    5021  156.19  5030.6  157.15  5036.5  155.85  5042.6   161.5  5051.9  162.18
  5057.8  163.94  5066.1  163.27  5073.2  164.66  5127.3   166.5  5189.4  169.23
  5204.8  168.83  5241.6  171.56  5279.4  172.37  5400.3  176.53  5470.7  177.82
#Mann= 7 ,-1 , 0
  4298.8     .07       0    4385     .12       0  4454.5      .1       0
    4973     .05       0  4978.9      .1       0  5127.3    .035       0
  5279.4     .12       0
Bank Sta=4973,4978.9
XS Rating Curve= 0 ,0
Exp/Cntr=0.3,0.1

Type RM Length L Ch R = 1 ,13100   ,143,143,143
BEGIN DESCRIPTION:
Mapping XS 2f1cc2a7
END DESCRIPTION:
XS GIS Cut Line= 3
      2524773.76      13509152.3      2524682.61     13508566.33
      2524535.53     13508228.91
#Sta/Elev= 30
  4416.1  174.44  4446.5  173.55  4546.7  170.04  4595.5  167.69  4646.9  166.31
  4757.5   162.4  4797.9  161.92  4808.1  161.32  4827.1  161.47  4909.3  160.22
  4949.7  161.29  4980.1  160.64  4990.2   159.2  5000.3  156.76  5004.1  153.69
  5004.6  153.19    5010  153.19  5010.5  153.69  5021.5  155.03  5039.3  159.09
  5062.7  160.94  5068.1   160.7  5086.1  162.88  5091.6  162.58  5108.7  163.32
  5206.9  164.11  5237.5  165.47  5266.4  165.67  5321.2   167.5  5377.2  171.13
#Mann= 7 ,-1 , 0
  4416.1     .07       0  4446.5     .12       0  4546.7     .05       0
  4646.9      .1       0  5004.1     .05       0  5010.5      .1       0
  5321.2     .12       0
Bank Sta=5004.1,5010.5
XS Rating Curve= 0 ,0
Exp/Cntr=0.3,0.1

Type RM Length L Ch R = 1 ,12957   ,164,164,164
BEGIN DESCRIPTION:
Mapping XS 231ebda2
END DESCRIPTION:
XS GIS Cut Line= 3
      2524856.22     13509126.24      2524825.83     13508540.29
      2524739.51     13508203.61
#Sta/Elev= 30
  4448.4  175.06  4479.7  173.52  4548.8  171.28  4589.8  169.94  4647.7  167.04
    4710  164.13  4860.2  159.57  4880.2  160.03  4910.3  159.96  4960.3  159.15
  4970.3  159.63  4980.3  158.59  4990.4  158.99  5007.2  152.97  5007.7  152.47
  5013.1  152.47  5013.6  152.97  5020.4  154.72  5030.3  158.18  5040.6  158.23
  5050.9   159.1  5057.4   160.2  5081.9  161.56  5092.2     162  5133.5  161.99
  5220.5  163.76  5319.7  167.61  5342.8  168.55  5350.3   169.4  5382.7  170.65
#Mann= 6 ,-1 , 0
  4448.4     .05       0  4548.8     .12       0  4647.7      .1       0
  5007.2     .05       0  5013.6      .1       0  5319.7     .12       0
Bank Sta=5007.2,5013.6
XS Rating Curve= 0 ,0
Exp/Cntr=0.3,0.1

Type RM Length L Ch R = 1 ,12793   ,350,350,350
BEGIN DESCRIPTION:
Mapping XS b39e765a
END DESCRIPTION:
XS GIS Cut Line= 4
      2524996.57     13509178.89      2524937.59     13508644.54
      2524991.37     13508486.67      2524817.88     13508160.51
#Sta/Elev= 30
  4377.4  177.19  4511.3  172.39  4627.1  168.25  4693.2  165.71  4723.4  163.94
  4773.7  162.39    4834  158.94  4864.2  159.11  4891.2  157.72  4912.2  158.88
  4952.5  158.34  4967.3  157.68  4989.1  155.81  4995.8   154.6  4996.3   154.1
  5001.7   154.1  5002.2   154.6  5009.6  155.14  5015.2  159.04  5020.5  161.35
    5109  160.49    5163  160.82  5235.2  162.81  5350.2  168.21  5361.3  168.83
    5367  168.66  5412.1   170.9  5427.3  171.18  5443.6  173.03  5451.2  173.35
#Mann= 6 ,-1 , 0
  4377.4     .05       0  4511.3     .07       0  4627.1      .1       0
  4995.8     .05       0  5002.2      .1       0  5350.2     .12       0
Bank Sta=4995.8,5002.2
XS Rating Curve= 0 ,0
Exp/Cntr=0.3,0.1

Type RM Length L Ch R = 1 ,12443   ,196,196,196
BEGIN DESCRIPTION:
JOHNS CREEK 21.0
END DESCRIPTION:
XS GIS Cut Line= 3
      2525208.22     13509151.13      2525213.43     13508661.89
      2524924.99     13508224.98
#Sta/Elev= 30
  4522.7  175.47  4565.3  174.46  4834.9  166.37  4898.8  163.87  4958.9  160.29
  4968.9     158  4978.9  157.16  4988.9  155.07  4998.9  151.08  5004.7  150.75
  5005.2  150.25  5010.7  150.25  5011.2  150.75    5012  150.75  5016.2  153.99
  5031.3  158.09    5046  158.76  5094.4  159.02  5116.1  160.22  5175.8  160.88
  5283.8  160.17  5341.3  160.39  5347.3  161.02  5362.4  161.28  5368.4  162.46
  5383.4  162.19  5449.7  164.09  5517.2  168.35  5527.9  168.33  5535.5  169.03
#Mann= 7 ,-1 , 0
  4522.7     .05       0  4565.3     .07       0  4834.9     .05       0
  5004.7     .05       0  5011.2     .05       0    5046      .1       0
  5517.2     .12       0
Bank Sta=5004.7,5011.2
XS Rating Curve= 0 ,0
Exp/Cntr=0.3,0.1

Type RM Length L Ch R = 1 ,12247   ,208,208,208
BEGIN DESCRIPTION:
JOHNS CREEK 20.0
END DESCRIPTION:
XS GIS Cut Line= 3
        2525375.       13508875.        2525375.       13508575.
      2524974.99     13508174.99
#Sta/Elev= 30
    4700  167.46  4731.4  166.71    4850  162.63    4870  161.38    4920  159.51
    4950  157.27    4970  154.61    4980  153.74  4986.8  151.42  4987.3  150.92
  4992.8  150.92  4993.3  151.42  4997.5  152.61  5003.5  152.61  5008.8  153.48
  5042.4  158.66  5056.6  159.68  5084.9  160.47  5169.7  159.58  5183.9  159.91
  5240.4  159.53  5339.4  159.85    5396   161.1    5470  165.41  5480.8  165.91
  5509.1  168.09  5537.4  169.16  5551.5  170.12  5562.2  171.54  5565.7  171.54
#Mann= 6 ,-1 , 0
    4700     .07       0  4731.4     .05       0  4986.8     .05       0
  4993.3     .05       0  5008.8      .1       0    5470     .07       0
Bank Sta=4986.8,4993.3
XS Rating Curve= 0 ,0
Exp/Cntr=0.3,0.1

Type RM Length L Ch R = 1 ,12039   ,235,235,235
BEGIN DESCRIPTION:
Mapping XS f23de02e
END DESCRIPTION:
XS GIS Cut Line= 3
      2525646.14     13508904.85      2525546.32      13508466.5
      2525125.56     13508019.71
#Sta/Elev= 30
  4541.1  166.86  4596.5  166.68  4858.9  163.64  4889.7  161.82  4932.4  157.21
  4975.5  155.56    4982   152.1  4985.6  151.15  4986.1  150.65  4992.1  151.15
  4999.7  151.96  5006.6  154.85  5013.9  156.64  5020.8  156.75  5028.1  158.24
  5034.9  157.57  5063.3  159.08  5095.6  159.03  5127.2  160.22  5141.4  159.48
  5212.2  158.75  5254.2  159.41  5296.7  159.01  5346.5  159.85  5353.4  160.53
  5367.5     160  5493.1  165.64  5544.3  171.96  5551.6  171.96  5604.4  175.99
#Mann= 6 ,-1 , 0
  4541.1     .05       0  4596.5     .07       0  4985.6     .05       0
  4992.1     .07       0  5095.6      .1       0  5493.1     .07       0
Bank Sta=4985.6,4992.1
XS Rating Curve= 0 ,0
Exp/Cntr=0.3,0.1

Type RM Length L Ch R = 1 ,11804   ,487,487,487
BEGIN DESCRIPTION:
JOHNS CREEK 19.0
END DESCRIPTION:
XS GIS Cut Line= 3
      2525875.01     13508925.05        2525725.       13508325.
      2525375.01     13507925.02
#Sta/Elev= 30
  4381.8  167.78  4433.4  166.34  4487.5  166.42  4523.6  164.63  4629.2  163.18
  4652.5   161.7  4670.6  162.61  4734.9  161.94  4776.1  163.55  4804.5  161.45
  4879.4  160.91  4894.7  161.13  4928.2  155.85  4959.1  154.27  4973.9  152.19
  4974.4  151.69  4980.4  152.19    4990  153.95  5003.3  154.43  5028.3   157.4
  5078.6  158.47  5199.2  155.44  5234.3   156.5  5240.9  157.91    5277  154.32
  5297.9  158.11  5361.5  161.31  5432.6  167.48  5489.3     171  5531.8  172.95
#Mann= 8 ,-1 , 0
  4381.8     .12       0  4652.5     .07       0  4670.6     .12       0
  4879.4     .07       0  4973.9     .05       0  4980.4     .07       0
  5003.3      .1       0  5489.3    .063       0
Bank Sta=4973.9,4980.4
XS Rating Curve= 0 ,0
Exp/Cntr=0.3,0.1

Type RM Length L Ch R = 1 ,11317   ,86,86,86
BEGIN DESCRIPTION:
Mapping XS 8b94ac91
END DESCRIPTION:
XS GIS Cut Line= 4
      2526401.92     13509178.72      2526033.01     13508783.77
      2525750.89     13508024.22      2525481.77     13507742.08
#Sta/Elev= 30
  3631.1  178.09  3900.3  171.06  3985.3  167.68    4063  167.25  4246.5  163.21
  4404.8  160.38  4435.1  161.23  4479.6  159.38  4628.8  159.73  4660.9  160.28
  4724.8  157.52  4728.1  156.72  4735.6  158.34  4771.3  158.25  4906.3  158.17
    4949  156.48    4955  157.64  4978.7  152.27  4996.2  149.83  4996.7  149.33
  5002.8  149.83  5006.8  151.29  5027.8   153.3  5063.3  162.93  5084.4  166.79
  5133.8  170.16    5141  174.02  5155.2  175.27  5231.5  175.03  5371.7   175.2
#Mann= 9 ,-1 , 0
  3631.1     .05       0  4246.5     .12       0  4628.8     .07       0
  4724.8     .12       0  4771.3      .1       0  4996.2     .05       0
  5002.8      .1       0  5063.3    .063       0  5231.5    .094       0
Bank Sta=4996.2,5002.8
XS Rating Curve= 0 ,0
Exp/Cntr=0.3,0.1

Type RM Length L Ch R = 1 ,11231   ,317,317,317
BEGIN DESCRIPTION:
Mapping XS 1832a1a6
END DESCRIPTION:
XS GIS Cut Line= 3
      2526471.36     13509165.69      2526089.43     13508488.63
      2525668.43      13507707.4
#Sta/Elev= 30
  3637.7  178.74  3879.3  171.11    3885  172.15  3900.9  167.37    3914  166.91
  4143.6  167.12  4165.3  166.79    4171  165.23  4201.1  163.61  4384.8  160.07
  4437.3  159.68  4551.1  157.79  4657.7  157.88  4692.7  159.08  4790.8  157.49
  4878.4  159.04  4900.3  157.72  4961.5  157.45  4975.8  156.61  4984.6  149.48
  4985.1  148.98  4991.2  149.48  5042.3  156.67  5069.8  162.22  5146.1  167.54
  5158.5  170.45    5168  170.36  5173.7  173.56  5216.7  175.44  5302.5  175.26
#Mann= 9 ,-1 , 0
  3637.7     .05       0  4384.8     .12       0  4437.3      .1       0
  4551.1     .12       0  4961.5      .1       0  4984.6     .05       0
  4991.2      .1       0  5158.5    .063       0  5216.7    .094       0
Bank Sta=4984.6,4991.2
XS Rating Curve= 0 ,0
Exp/Cntr=0.3,0.1

Type RM Length L Ch R = 1 ,10914   ,713,713,713
BEGIN DESCRIPTION:
JOHNS CREEK 17.0
END DESCRIPTION:
XS GIS Cut Line= 3
      2526475.01     13509025.04        2526075.       13507825.
        2526075.     13507624.95
#Sta/Elev= 30
  3738.6  174.56  3865.1  170.63  3949.5  169.14  4012.7  166.67  4118.4  166.94
  4160.3  166.55  4170.8  164.57    4213  162.22  4328.9  160.64    4350  161.63
  4381.6  160.81  4392.2  159.38  4443.8  158.57  4476.5  157.63  4581.9   156.8
  4613.5  155.72  4634.6  156.37  4782.2  157.02  4877.1  155.31  4919.2  155.79
  4947.8  153.96  4961.4  150.87  4979.1  148.92  4979.6  148.42  4985.8  148.92
    4993  154.15  5000.9     157  5049.8  159.49  5143.6  164.61  5203.6  165.97
#Mann= 7 ,-1 , 0
  3738.6     .05       0  4118.4     .07       0  4443.8      .1       0
  4947.8     .07       0  4979.1     .05       0  4985.8     .07       0
  5049.8     .12       0
Bank Sta=4979.1,4985.8
XS Rating Curve= 0 ,0
Exp/Cntr=0.3,0.1

Type RM Length L Ch R = 1 ,10201   ,206,206,206
BEGIN DESCRIPTION:
Mapping XS be564cd2
END DESCRIPTION:
XS GIS Cut Line= 4
      2526753.79     13508585.41      2526654.83     13508163.54
      2526607.96     13508064.59      2526180.87     13507606.24
#Sta/Elev= 30
  4578.9  166.42  4722.4  165.44  4753.9  163.94  4814.5   163.2  4866.9  163.74
  4897.3  161.91    4950  160.66  4969.6  158.07  4987.3  151.69  4992.5  152.03
  5005.4  145.62  5005.9  145.12  5012.3  145.62  5019.8  147.55  5025.4  147.29
  5032.7  150.18  5042.6  151.86  5088.1  153.92  5113.6  152.79  5144.9  154.49
  5233.8  155.25  5251.5  155.46    5350  156.13  5392.6  155.27  5413.6  156.63
  5427.7  155.65  5459.5  156.14  5597.7   157.1  5682.3  159.83  5748.2  163.42
#Mann= 8 ,-1 , 0
  4578.9     .07       0  4814.5     .05       0  5005.4     .05       0
  5012.3     .05       0  5113.6     .12       0  5233.8     .05       0
  5251.5      .1       0  5459.5     .07       0
Bank Sta=5005.4,5012.3
XS Rating Curve= 0 ,0
Exp/Cntr=0.3,0.1

Type RM Length L Ch R = 1 ,9995    ,677,677,677
BEGIN DESCRIPTION:
JOHNS CREEK 16.0
END DESCRIPTION:
XS GIS Cut Line= 3
      2526874.98     13508174.97        2526825.       13508075.
      2526074.99     13507374.99
#Sta/Elev= 30
  4888.5  163.58  4896.4  163.36  4924.8  162.88  4941.6  160.94  4947.2  157.89
  4955.5  151.35  4963.9  146.31  4974.5  146.11    4975  145.61  4981.4  146.11
  4991.9  149.38  5003.7  150.08  5014.2  152.14  5042.5  153.37  5078.2  152.12
  5086.7  152.68  5106.5  153.39  5127.5  152.95  5177.4  154.61    5224  154.42
  5367.3  155.21  5424.6  154.44  5559.4  155.44  5615.8  157.43  5728.9  159.38
  5813.9  163.32  5842.2  166.86  5867.8  167.82  5983.9  171.47  6026.2  171.78
#Mann= 8 ,-1 , 0
  4888.5     .12       0  4896.4     .05       0  4974.5     .05       0
  4981.4     .05       0  5086.7     .12       0    5224     .05       0
  5367.3     .07       0  5867.8     .05       0
Bank Sta=4974.5,4981.4
XS Rating Curve= 0 ,0
Exp/Cntr=0.3,0.1

Type RM Length L Ch R = 1 ,9318    ,682,682,682
BEGIN DESCRIPTION:
Mapping XS aa3b2feb
END DESCRIPTION:
XS GIS Cut Line= 4
      2527578.14     13508492.96      2527035.61     13507737.76
       2526549.5     13507433.94      2525951.44     13507169.58
#Sta/Elev= 30
  3726.1  166.03  3874.9  162.99  3950.9  160.74  4037.1  160.29  4070.1  161.39
  4114.3   160.1  4292.3  159.94    4487  157.48  4558.7   155.3  4573.2  156.13
  4594.3  154.21  4644.7  153.38  4716.3  153.46  4911.1  150.61  4955.5  149.72
  4970.8  146.85  4995.2  144.83  4995.7  144.33  5002.2  144.83  5007.4  146.56
  5013.3  145.71  5018.7  147.16  5028.6  150.49  5071.1  150.13  5128.9   155.9
  5224.4  157.35  5398.1  161.39  5511.6  166.83  5573.1  169.93  5883.1  176.65
#Mann= 11 ,-1 , 0
  3726.1     .07       0  3874.9     .12       0  3950.9     .07       0
  4037.1     .12       0  4716.3     .05       0  4911.1     .07       0
  4995.2     .05       0  5002.2     .07       0  5018.7     .12       0
  5224.4     .07       0  5511.6     .05       0
Bank Sta=4995.2,5002.2
XS Rating Curve= 0 ,0
Exp/Cntr=0.3,0.1

Type RM Length L Ch R = 1 ,8636    ,448,448,448
BEGIN DESCRIPTION:
JOHNS CREEK 14.0
END DESCRIPTION:
XS GIS Cut Line= 3
      2527508.12      13508058.5        2527325.       13507375.
        2527075.       13506975.
#Sta/Elev= 30
  4296.3  157.69  4324.3  157.24  4462.7  153.83  4475.9  153.69  4486.8   152.3
    4507  153.06    4546  152.86  4601.7  152.84  4631.2  151.69  4668.1  151.62
  4751.7   151.3  4786.4  152.67  4826.4  152.41  4866.4  149.92  4941.3   148.9
  4977.7  143.02  4978.2  142.52  4984.9  143.02  5026.9  145.68  5032.8  145.16
    5054  145.87  5069.4  148.07  5084.7  148.63  5098.2   151.7  5187.1  153.24
    5228  153.39  5309.9  155.84  5315.8  155.26  5450.4  157.63  5475.6  157.83
#Mann= 10 ,-1 , 0
  4296.3     .07       0  4324.3     .05       0  4462.7     .12       0
    4546     .05       0  4668.1     .12       0  4751.7      .1       0
  4977.7     .05       0  4984.9      .1       0  5187.1     .07       0
  5450.4     .05       0
Bank Sta=4977.7,4984.9
XS Rating Curve= 0 ,0
Exp/Cntr=0.3,0.1

Type RM Length L Ch R = 1 ,8188    ,601,601,601
BEGIN DESCRIPTION:
JOHNS CREEK 13.0
END DESCRIPTION:
XS GIS Cut Line= 3
      2527824.98     13507674.95        2527725.       13507425.
      2527475.01     13507125.02
#Sta/Elev= 30
  4730.4  154.22    4799   152.9  4860.7  148.91  4936.3  148.49  4967.3  149.35
  4978.1  146.61  4984.8  142.76  4990.2  142.97  4993.3  139.36  4993.8  138.86
  5000.1  138.86  5000.6  139.36  5002.9  139.36  5006.8  141.05  5013.3  142.58
  5021.1  146.51  5049.7  147.81  5078.6  147.97  5113.5  147.32  5134.3  148.53
  5169.5  148.27  5191.6  146.48  5226.8   144.7  5233.9  145.66  5241.1  148.86
  5255.4  151.35  5290.5  152.69  5319.2  152.81  5325.7  153.46  5390.1  154.05
#Mann= 5 ,-1 , 0
  4730.4     .07       0  4860.7     .05       0  4993.3     .05       0
  5000.6     .05       0  5078.6     .07       0
Bank Sta=4993.3,5000.6
XS Rating Curve= 0 ,0
Exp/Cntr=0.3,0.1

Type RM Length L Ch R = 1 ,7587    ,319,319,319
BEGIN DESCRIPTION:
Mapping XS c70f4545
END DESCRIPTION:
XS GIS Cut Line= 3
      2528094.93     13507565.99      2528029.83     13507214.47
      2527488.67     13506868.12
#Sta/Elev= 30
  4428.4  155.61  4455.1  155.06  4555.9  150.82  4671.8  147.51  4724.3  148.31
  4729.7  147.63    4765  147.17  4775.2  146.63  4795.9  143.93  4811.1  144.59
  4862.7  144.16  4883.8  144.83    4905  143.03  4920.2  143.82  4962.5  142.56
  4977.7  143.32  5001.6  139.96  5002.1  139.46    5009  139.96    5014  142.24
  5035.2  144.63  5060.8  143.91  5101.1  144.03  5135.9  142.52  5165.4  145.57
  5180.6  149.16  5201.8   150.3  5244.1  150.49    5332  153.09  5428.4  154.34
#Mann= 7 ,-1 , 0
  4428.4     .07       0  4455.1     .12       0  4555.9     .07       0
  5001.6     .05       0    5009     .07       0  5060.8     .05       0
  5101.1     .07       0
Bank Sta=5001.6,5009
XS Rating Curve= 0 ,0
Exp/Cntr=0.3,0.1

Type RM Length L Ch R = 1 ,7268    ,191,191,191
BEGIN DESCRIPTION:
JOHNS CREEK 12.0
END DESCRIPTION:
XS GIS Cut Line= 3
        2528225.     13507425.01        2528125.       13507075.
      2527725.01     13506725.01
#Sta/Elev= 30
  4631.5  154.21  4687.4  151.98  4745.9  147.61  4787.5  147.11  4827.8  147.73
  4922.7  147.44  4933.1  146.55  4939.6  145.27  4944.8  142.45  4953.9  139.67
  4981.4  136.66  4981.9  136.16  4988.3  136.16  4988.8  136.66  4998.8  136.87
  5002.6  139.71  5016.9  143.06  5031.1   144.1  5059.6  144.48  5066.2  145.58
  5073.8  145.73  5080.5  146.84  5088.1  147.28  5108.9  147.68  5194.4  146.71
  5250.3  148.35  5293.1  147.85  5347.6  149.13  5515.1  151.61    5527  152.08
#Mann= 5 ,-1 , 0
  4631.5     .07       0  4981.4     .05       0  4988.8     .07       0
  5347.6     .05       0  5515.1     .07       0
Bank Sta=4981.4,4988.8
XS Rating Curve= 0 ,0
Exp/Cntr=0.3,0.1

Type RM Length L Ch R = 1 ,7077    ,708,708,708
BEGIN DESCRIPTION:
Mapping XS 642fe4c1
END DESCRIPTION:
XS GIS Cut Line= 4
      2528645.85     13507703.04      2528329.01     13507151.82
       2528068.6     13506557.21      2527735.48     13506319.26
#Sta/Elev= 30
  4112.7  156.64    4244  154.05  4259.8  154.51  4330.2  153.11  4404.7  153.09
    4517  151.68  4592.7  150.21  4632.6  148.63    4668   146.4  4748.2  146.83
  4788.1   146.1  4823.9  145.76  4857.1  144.07  4870.6  143.47  4908.8  144.93
  4930.6  144.34  4998.4  139.69  5012.6  136.46  5013.1  135.96  5020.1  136.46
  5021.8   136.7  5028.9  141.45  5039.7  144.84  5045.2  143.89    5074  146.13
  5097.4  146.29  5249.3  145.89  5383.7  148.81  5557.9   154.2    5807  161.23
#Mann= 13 ,-1 , 0
  4112.7     .05       0  4404.7     .07       0    4517     .05       0
  4592.7     .07       0  4632.6     .12       0  4748.2     .07       0
  4788.1     .12       0  4857.1     .07       0  5012.6     .05       0
  5020.1     .07       0  5249.3      .1       0  5383.7     .12       0
  5557.9     .05       0
Bank Sta=5012.6,5020.1
XS Rating Curve= 0 ,0
Exp/Cntr=0.3,0.1

Type RM Length L Ch R = 1 ,6369    ,288,288,288
BEGIN DESCRIPTION:
Mapping XS fbe02e39
END DESCRIPTION:
XS GIS Cut Line= 3
      2529813.41     13507872.33      2528719.64     13506991.23
      2527829.97     13506136.28
#Sta/Elev= 30
  3587.4  154.94  3890.6  152.46  4135.6   147.5  4263.5  144.83  4382.3  144.45
  4386.9   144.6  4510.4  144.32  4545.2  144.39  4825.4  144.56  4935.1     145
  4943.1  146.45    4985  136.05  4995.7   135.5  4996.2     135  5003.2   135.5
  5005.1  135.95  5070.2  139.41  5077.5  141.03  5137.9  141.85  5233.1  145.57
  5275.6  145.43  5331.9  142.24  5480.6   146.3  5664.3  147.35  5756.4  149.31
  5818.3  152.56  5909.1  156.12  6032.2   159.7  6039.1  162.15  6225.8  166.78
#Mann= 14 ,-1 , 0
  3587.4     .05       0  4135.6    .035       0  4263.5     .05       0
  4382.3    .035       0  4386.9     .12       0  4510.4     .05       0
  4545.2     .12       0  4825.4     .07       0  4995.7     .05       0
  5003.2     .07       0  5005.1     .12       0  5137.9      .1       0
  5818.3     .12       0  5909.1     .05       0
Bank Sta=4995.7,5003.2
XS Rating Curve= 0 ,0
Exp/Cntr=0.3,0.1

Type RM Length L Ch R = 1 ,6081    ,1090,1090,1090
BEGIN DESCRIPTION:
Mapping XS 10a49a7d
END DESCRIPTION:
XS GIS Cut Line= 3
      2529874.15     13507776.82      2528854.19     13506765.54
      2528363.74     13506196.96
#Sta/Elev= 30
  3575.1  153.44  3704.1  154.48  3712.8  154.31  3816.2  150.94  3853.5   152.2
    4111  146.93  4136.5  146.29  4210.1  143.83  4318.3  142.04  4339.5  138.57
  4417.3  143.13  4598.9  142.82  4692.7  142.71  4933.4  143.16  5001.2  136.02
  5014.4  132.05  5014.9  131.55  5022.2  132.05  5032.5  137.55  5061.1  141.06
  5081.9   140.5  5124.7  146.72  5158.1  146.77  5262.9   150.8  5412.2  154.46
  5458.2  156.38  5611.9  154.11  5649.1  153.03  5656.7  155.39  5762.3  153.35
#Mann= 16 ,-1 , 0
  3575.1    .035       0  3704.1     .05       0  3712.8    .035       0
  3853.5     .05       0    4111    .035       0  4136.5     .07       0
  4210.1      .1       0  4598.9     .12       0  4692.7      .1       0
  5001.2     .12       0  5014.4     .05       0  5022.2     .12       0
  5158.1    .035       0  5262.9     .12       0  5412.2     .05       0
  5611.9     .12       0
Bank Sta=5014.4,5022.2
XS Rating Curve= 0 ,0
Exp/Cntr=0.3,0.1

Type RM Length L Ch R = 1 ,4991    ,1101,1101,1101
BEGIN DESCRIPTION:
Mapping XS f6e0bd62
END DESCRIPTION:
XS GIS Cut Line= 3
      2529969.64     13507815.89       2529587.7     13506808.94
      2528638.61     13505885.86
#Sta/Elev= 30
  4151.3  153.61  4208.9  155.33  4258.5  152.04    4286  152.64  4426.4  150.63
  4581.9  149.52  4780.9  146.56  4908.9  142.23  4939.1  136.06  4986.5  133.63
  5003.8  130.79  5004.3  130.29  5011.9  130.79  5029.5  138.49  5132.2  140.18
  5196.4  140.44  5251.5  141.04  5345.3   140.5  5445.1  140.14  5598.8   145.7
  5688.4  151.46  5745.8  154.97    5834  159.16  5879.3   160.6  5968.5  164.45
  5989.6  167.62    6131  171.51  6293.6   170.3  6549.2   163.8  6552.2  163.73
#Mann= 17 ,-1 , 0
  4151.3    .035       0    4286     .05       0  4426.4    .035       0
  4581.9     .07       0  4780.9      .1       0  5003.8     .05       0
  5011.9      .1       0  5132.2     .07       0  5196.4     .12       0
  5251.5     .07       0  5345.3     .12       0  5598.8      .1       0
  5688.4    .035       0  5745.8     .07       0    5834     .12       0
  5879.3     .05       0  6549.2     .12       0
Bank Sta=5003.8,5011.9
XS Rating Curve= 0 ,0
Exp/Cntr=0.3,0.1

Type RM Length L Ch R = 1 ,3890    ,664,664,664
BEGIN DESCRIPTION:
Mapping XS a3af5c6f
END DESCRIPTION:
XS GIS Cut Line= 4
      2530138.91     13507763.82       2530030.4      13506405.3
      2528997.42     13506140.54      2528619.89     13505680.56
#Sta/Elev= 30
  3477.1  152.63  3545.3  151.96  3907.3  148.05  4040.9  144.79    4140  142.85
  4167.9  142.81  4338.3  142.08  4669.7  137.14  4833.9  137.97  4873.4  138.29
  4959.1  137.98  4983.5  130.88    4986  128.03  4986.5  127.53  4994.1  128.03
  5024.3  131.61  5068.1  131.94  5124.3  137.29  5168.9  138.59  5258.5  138.16
  5269.7  140.47  5370.4  143.64  5462.6  152.63    5572  159.41  5672.7  163.28
  5705.2  164.59  5805.6  169.09  5939.8  171.82  6377.6  165.43  6501.4   163.5
#Mann= 18 ,-1 , 0
  3477.1    .035       0  3545.3     .05       0  4040.9    .035       0
    4140     .05       0  4167.9     .07       0  4338.3     .12       0
  4833.9     .07       0  4873.4     .12       0    4986     .05       0
  4994.1     .12       0  5068.1      .1       0  5168.9    .035       0
  5269.7     .12       0  5370.4     .07       0    5572     .05       0
  5672.7     .07       0  5705.2     .05       0  6377.6    .035       0
Bank Sta=4986,4994.1
XS Rating Curve= 0 ,0
Exp/Cntr=0.3,0.1

Type RM Length L Ch R = 1 ,3226    ,836,836,836
BEGIN DESCRIPTION:
Mapping XS 5a855827
END DESCRIPTION:
XS GIS Cut Line= 3
      2530282.14     13507516.41       2530030.4       13505802.
      2529205.77     13505246.46
#Sta/Elev= 30
  3243.8  149.38  3657.8  142.51    3743  142.68  3757.9  141.19  3857.9  140.05
  4158.1  136.02  4458.1  137.56  4478.3  139.89  4622.6  138.51  4660.2   135.5
  4710.8  137.38  4758.5  136.61    4822  133.61  4858.6  134.02  4902.8  134.64
  4976.6  132.26  4984.7  129.15  5003.1  126.63  5003.6  126.13  5011.3  126.63
  5029.6  131.06  5035.6  136.82  5043.4  139.28  5109.7  139.92    5220  141.75
  5311.8  143.89    5496  148.89  5680.2   158.4  5769.2  161.34  5970.9  165.67
#Mann= 16 ,-1 , 0
  3243.8     .05       0  3657.8    .035       0  3757.9     .05       0
  3857.9     .12       0  4158.1     .07       0  4622.6     .12       0
  4758.5     .07       0  4858.6      .1       0  5003.1     .05       0
  5011.3      .1       0  5109.7    .035       0    5220      .1       0
  5311.8     .12       0    5496     .07       0  5680.2     .12       0
  5769.2    .035       0
Bank Sta=5003.1,5011.3
XS Rating Curve= 0 ,0
Exp/Cntr=0.3,0.1

Type RM Length L Ch R = 1 ,2390    ,517,517,517
BEGIN DESCRIPTION:
Mapping XS 633f9b45
END DESCRIPTION:
XS GIS Cut Line= 3
      2531134.57     13507420.04      2530641.51     13506093.66
      2529815.12     13505111.02
#Sta/Elev= 30
  3564.4  143.35  3825.8  141.37  4206.7  135.31  4565.9  133.09  4743.3  133.55
  4756.8  135.93  4867.5   137.3  4938.8  135.41  4958.6  132.46  4976.1  126.07
  4979.5  126.07  4986.7  122.19  4987.2  121.69  4994.9  122.19  5011.6  127.03
  5061.1  133.73  5090.9  135.46    5178  138.81  5191.1     139  5323.1  138.26
  5332.9  137.72    5455  137.19  5480.7  137.11    5587  137.17  5628.6  136.94
  5718.9  136.82  5819.8  136.84  5997.6  138.61  6246.7  145.07  6263.4  145.51
#Mann= 17 ,-1 , 0
  3564.4     .05       0  4565.9      .1       0  4938.8     .12       0
  4986.7     .05       0  4994.9     .12       0  5090.9      .1       0
    5178     .12       0  5191.1      .1       0  5323.1     .12       0
  5332.9      .1       0    5455    .035       0  5480.7     .07       0
    5587    .035       0  5628.6      .1       0  5718.9    .035       0
  5819.8     .12       0  6246.7     .07       0
Bank Sta=4986.7,4994.9
XS Rating Curve= 0 ,0
Exp/Cntr=0.3,0.1

Type RM Length L Ch R = 1 ,1873    ,415,415,415
BEGIN DESCRIPTION:
Mapping XS c008bb6c
END DESCRIPTION:
XS GIS Cut Line= 3
      2531547.77     13507284.64      2531110.26     13506048.52
      2530144.96     13504985.99
#Sta/Elev= 30
  3682.9  144.41  3762.9  143.13  4043.2  138.25  4552.4  134.69  4700.9  134.99
  4711.5  136.88  4726.3  137.05  4889.8  136.51  4942.8  134.92  4968.2  134.25
  4976.7  131.89  4993.4  122.95  5017.5  122.03    5018  121.53    5026  122.03
  5035.9  125.95  5042.7  126.32  5050.1  128.73  5078.5  131.57  5134.6  131.23
  5190.9  133.68  5269.3  136.53  5325.8  138.42  5368.4  138.69  5556.5  137.62
  5793.4  134.94  5863.7  135.74  5948.9  135.12  6267.8  136.64  6429.7  139.27
#Mann= 9 ,-1 , 0
  3682.9     .12       0  3762.9     .05       0  4889.8     .07       0
  4942.8     .12       0  5017.5     .05       0    5026     .12       0
  5190.9      .1       0  5269.3     .07       0  5556.5     .12       0
Bank Sta=5017.5,5026
XS Rating Curve= 0 ,0
Exp/Cntr=0.3,0.1
