--- TRIB 3 TO YORKTOWN CREEK.prj (project) ---

Proj Title=TRIB 3 TO YORKTOWN CREEK Base Level Engineering
Current Plan=p01
Default Exp/Contr=0.3,0.1
English Units
Geom File=g01
Flow File=f01
Plan File=p01
BEGIN DESCRIPTION:
TRIB 3 TO YORKTOWN CREEK
END DESCRIPTION:

--- TRIB 3 TO YORKTOWN CREEK.p01 (plan) ---

Plan Title=Multiple Run
Short Identifier=Multiple
Geom File=g01
Flow File=f01
Subcritical Flow
K Sum by GR= 0
Std Step Tol= 0.01
Critical Tol= 0.01
Num of Std Step Trials= 20
Max Error Tol= 0.3
Flow Tol Ratio= 0.001
Split Flow NTrial= 30
Split Flow Tol= 0.02
Split Flow Ratio= 0.02
Log Output Level= 0
Friction Slope Method= 1
Unsteady Friction Slope Method= 2
Unsteady Bridges Friction Slope Method= 1
Parabolic Critical Depth
Global Vel Dist=  1 , 1 , 1
Global Log Level= 0
CheckData=True
Encroach Param= -1, 0, 0, 0
BEGIN DESCRIPTION:
Multiple Run
END DESCRIPTION:

--- TRIB 3 TO YORKTOWN CREEK.f01 (steady flow) ---

Flow Title=Multiple
Number of Profiles=7
Profile Names=10-year,25-year,50-year,1pct_min,100-year,1pct_plu,500-year
River Rch & RM= TRIB 3 TO YORKTO,Reach-1,24099
     243     371     480     303     604    1205     944
River Rch & RM= TRIB 3 TO YORKTO,Reach-1,22377
     429     681     904     583    1164    2323    1908
River Rch & RM= TRIB 3 TO YORKTO,Reach-1,20120
     651    1058    1427     933    1862    3715    3138
River Rch & RM= TRIB 3 TO YORKTO,Reach-1,16945
     878    1449    1977    1305    2604    5196    4479
River Rch & RM= TRIB 3 TO YORKTO,Reach-1,15437
    1017    1689    2312    1530    3053    6092    5281
River Rch & RM= TRIB 3 TO YORKTO,Reach-1,10408
    1826    3109    4325    2903    5791   11555   10289
River Rch & RM= TRIB 3 TO YORKTO,Reach-1,5360
    1886    3216    4481    3010    6006   11984   10695
River Rch & RM= TRIB 3 TO YORKTO,Reach-1,3283
    2240    3846    5383    3631    7245   14456   13008
Boundary for River Rch & Prof#=TRIB 3 TO YORKTO,Reach-1,1
Up Type=0
Dn Type=3
Dn Slope=0.005
Boundary for River Rch & Prof#=TRIB 3 TO YORKTO,Reach-1,2
Up Type=0
Dn Type=3
Dn Slope=0.005
Boundary for River Rch & Prof#=TRIB 3 TO YORKTO,Reach-1,3
Up Type=0
Dn Type=3
Dn Slope=0.005
Boundary for River Rch & Prof#=TRIB 3 TO YORKTO,Reach-1,4
Up Type=0
Dn Type=3
Dn Slope=0.005
Boundary for River Rch & Prof#=TRIB 3 TO YORKTO,Reach-1,5
Up Type=0
Dn Type=3
Dn Slope=0.005
Boundary for River Rch & Prof#=TRIB 3 TO YORKTO,Reach-1,6
Up Type=0
Dn Type=3
Dn Slope=0.005
Boundary for River Rch & Prof#=TRIB 3 TO YORKTO,Reach-1,7
Up Type=0
Dn Type=3
Dn Slope=0.005

--- TRIB 3 TO YORKTOWN CREEK.g01 (geometry) ---

Geom Title=Existing Conditions

River Reach=TRIB 3 TO YORKTO,Reach-1
Reach XY= 30
      2427825.00     13556225.00      2428266.54     13556321.50
      2428971.33     13555532.69      2429414.50     13555623.78
      2429780.86     13555377.07      2430884.81     13555214.49
      2431680.25     13554030.44      2432298.83     13553702.01
      2432915.32     13552785.17      2433261.55     13552788.63
      2433501.14     13551948.06      2434531.19     13551567.19
      2435568.29     13550584.16      2436038.34     13550561.59
      2436288.26     13550061.35      2436669.64     13549827.70
      2436732.62     13549168.49      2437081.80     13549117.14
      2437172.30     13548880.36      2438345.17     13548724.54
      2439354.97     13548924.94      2439873.28     13548871.66
      2440085.30     13548625.59      2441118.95     13548573.33
      2441516.86     13548281.06      2441808.33     13547591.65
      2442627.55     13547369.27      2442972.55     13546930.46
      2443814.45     13547123.91      2444925.00     13546575.00

Type RM Length L Ch R = 1,24099,179,179,179
BEGIN DESCRIPTION:
Mapping XS 3013f516
END DESCRIPTION:
XS GIS Cut Line= 4
      2427889.61     13556564.83      2427976.66     13556353.44
      2427949.30     13556191.78      2427844.85     13555885.89
#Sta/Elev= 30
  4785.6  377.22  4788.7  376.80  4796.2  376.60  4842.0  376.29  4866.0  374.71
  4889.9  374.79  4895.3  373.90  4904.4  373.25  4926.0  372.28  4943.2  372.32
  4996.5  370.64  5008.7  370.61  5008.9  370.11  5012.4  370.11  5012.7  370.61
  5038.4  370.94  5116.6  372.41  5176.1  374.56  5185.3  374.55  5235.4  376.64
  5266.7  377.61  5291.0  377.82  5298.0  378.37  5343.8  379.18  5354.4  378.91
  5360.7  379.30  5392.0  379.51  5480.7  381.13  5486.0  381.48  5501.4  381.50
#Mann=4,-1,0
  4785.6    0.04       0  5008.7    0.04       0  5012.7    0.04       0
  5038.4    0.05       0
Bank Sta=5008.7,5012.7
Exp/Cntr=0.3,0.1

Type RM Length L Ch R = 1,23920,332,332,332
BEGIN DESCRIPTION:
Mapping XS e10c8d0b
END DESCRIPTION:
XS GIS Cut Line= 4
      2427946.83     13556689.16      2428120.90     13556450.43
      2428135.82     13556134.58      2427986.58     13555910.72
#Sta/Elev= 30
  4629.8  377.15  4652.8  376.36  4682.2  376.13  4688.4  375.02  4696.8  374.71
  4703.0  373.78  4732.4  373.79  4738.6  372.33  4859.9  370.07  4868.4  370.33
  4889.2  369.80  4895.4  369.27  4924.5  369.01  4968.7  367.84  4969.0  367.34
  4972.5  367.34  4972.7  367.84  5080.9  368.80  5126.2  369.71  5249.5  371.77
  5277.0  372.90  5336.6  374.19  5349.1  374.96  5357.6  374.86  5372.6  375.60
  5452.2  377.44  5465.8  377.39  5474.3  377.83  5493.3  378.10  5510.5  378.97
#Mann=6,-1,0
  4629.8    0.04       0  4968.7    0.04       0  4972.7    0.04       0
  5126.2    0.05       0  5452.2    0.04       0  5474.3    0.05       0
Bank Sta=4968.7,4972.7
Exp/Cntr=0.3,0.1

Type RM Length L Ch R = 1,23588,229,229,229
BEGIN DESCRIPTION:
Mapping XS bebe33ce
END DESCRIPTION:
XS GIS Cut Line= 3
      2428434.26     13556709.08      2428349.70     13556194.27
      2428193.01     13555915.72
#Sta/Elev= 30
  4447.2  372.76  4499.6  371.44  4597.6  369.54  4613.5  368.35  4626.0  369.93
  4633.7  370.67  4653.8  367.89  4658.8  369.63  4674.3  367.04  4694.5  367.78
  4799.8  366.85  4906.1  366.11  4992.7  365.58  5036.9  367.01  5046.3  365.73
  5065.9  365.45  5066.2  364.95  5069.9  365.45  5110.9  366.07  5127.2  365.89
  5133.0  366.86  5140.2  366.31  5154.6  367.56  5192.2  366.51  5213.9  370.32
  5243.4  370.46  5266.4  371.71  5278.9  374.05  5286.0  376.79  5288.5  376.79
#Mann=8,-1,0
  4447.2    0.05       0  4499.6    0.04       0  4626.0    0.05       0
  4799.8    0.04       0  4906.1    0.05       0  5065.9    0.05       0
  5069.9    0.05       0  5110.9    0.04       0
Bank Sta=5065.9,5069.9
Exp/Cntr=0.3,0.1

Type RM Length L Ch R = 1,23359,315,315,315
BEGIN DESCRIPTION:
Mapping XS 6d027c2b
END DESCRIPTION:
XS GIS Cut Line= 3
      2428625.74     13556701.56      2428498.92     13556067.44
      2428327.33     13555826.22
#Sta/Elev= 30
  4243.1  375.96  4375.8  372.42  4433.4  370.45  4453.8  369.06  4477.8  370.77
  4484.3  370.18  4504.7  366.75  4552.7  366.86  4590.9  366.57  4681.8  365.42
  4820.9  365.06  4829.6  364.76  4832.7  364.11  4833.0  363.61  4836.5  363.61
  4836.7  364.11  4929.6  364.89  5009.0  364.30  5038.5  366.15  5052.3  366.17
  5059.4  367.07  5080.3  364.69  5101.4  367.23  5116.0  368.03  5130.8  368.00
  5151.7  369.70  5160.3  370.93  5166.4  372.61  5183.5  378.86  5185.8  378.86
#Mann=5,-1,0
  4243.1    0.05       0  4552.7    0.04       0  4590.9    0.05       0
  4832.7    0.05       0  4836.7    0.05       0
Bank Sta=4832.7,4836.7
Exp/Cntr=0.3,0.1

Type RM Length L Ch R = 1,23044,312,312,312
BEGIN DESCRIPTION:
TRIB 3 TO YORKTOWN CREEK 43.0
END DESCRIPTION:
XS GIS Cut Line= 3
      2428975.02     13556425.04      2428675.00     13555875.00
      2428425.00     13555775.00
#Sta/Elev= 30
  4447.8  373.41  4559.4  371.29  4586.9  367.89  4736.7  366.50  4835.6  365.35
  4847.3  365.16  4891.6  365.24  4903.5  363.65  4935.3  363.81  4941.0  362.50
  4949.0  363.02  4984.6  362.27  4994.6  362.73  5058.6  362.20  5058.8  361.70
  5062.3  361.70  5062.6  362.20  5083.8  362.88  5089.1  364.72  5113.4  364.33
  5118.8  362.81  5155.6  362.33  5226.5  364.55  5260.4  367.61  5268.2  368.26
  5274.9  369.74  5299.2  372.13  5311.3  375.07  5334.2  378.60  5343.6  379.15
#Mann=8,-1,0
  4447.8    0.04       0  4736.7    0.05       0  4835.6    0.04       0
  4847.3    0.05       0  5058.6    0.05       0  5062.6    0.05       0
  5155.6    0.04       0  5260.4    0.05       0
Bank Sta=5058.6,5062.6
Exp/Cntr=0.3,0.1

Type RM Length L Ch R = 1,22732,355,355,355
BEGIN DESCRIPTION:
Mapping XS b80e8a15
END DESCRIPTION:
XS GIS Cut Line= 4
      2429055.99     13556348.43      2428968.95     13555793.87
      2428737.67     13555562.58      2428414.37     13555473.05
#Sta/Elev= 30
  4287.9  372.42  4412.8  370.41  4421.9  370.77  4514.1  368.37  4582.2  365.78
  4644.8  365.70  4717.5  364.73  4746.9  363.45  4797.5  362.43  4870.9  362.53
  4886.6  362.60  4900.7  361.80  4929.0  358.65  5026.0  358.39  5026.3  357.89
  5029.8  357.89  5030.0  358.39  5063.4  359.04  5077.5  361.31  5084.6  361.60
  5127.0  361.57  5141.2  362.34  5148.2  365.32  5155.0  364.30  5162.4  367.01
  5169.4  365.27  5174.7  367.19  5185.2  367.88  5209.0  367.79  5511.8  369.32
#Mann=7,-1,0
  4287.9    0.05       0  4421.9    0.04       0  4870.9    0.05       0
  5026.0    0.05       0  5030.0    0.05       0  5155.0    0.04       0
  5209.0    0.05       0
Bank Sta=5026,5030
Exp/Cntr=0.3,0.1

Type RM Length L Ch R = 1,22377,268,268,268
BEGIN DESCRIPTION:
Mapping XS d80e6edb
END DESCRIPTION:
XS GIS Cut Line= 4
      2429090.82     13556353.39      2429128.12     13555701.85
      2429105.74     13555480.51      2429026.16     13555134.83
#Sta/Elev= 30
  4219.7  371.74  4273.0  370.97  4348.3  369.97  4388.4  368.65  4428.4  368.30
  4448.5  367.51  4488.5  367.23  4514.2  366.35  4572.5  364.93  4658.8  363.08
  4698.9  362.82  4738.9  361.42  4838.9  359.00  4887.2  357.83  4986.6  356.17
  4997.8  356.01  4998.1  355.51  5001.6  355.51  5001.8  356.01  5060.1  356.63
  5090.0  358.23  5110.7  358.77  5138.5  360.54  5192.8  363.56  5251.6  366.14
  5367.2  368.61  5418.5  370.71  5433.1  370.88  5439.1  371.52  5449.5  371.83
#Mann=10,-1,0
  4219.7    0.05       0  4273.0    0.04       0  4514.2    0.05       0
  4572.5    0.04       0  4838.9    0.05       0  4887.2    0.04       0
  4986.6    0.05       0  4997.8    0.05       0  5001.8    0.05       0
  5138.5    0.04       0
Bank Sta=4997.8,5001.8
Exp/Cntr=0.3,0.1

Type RM Length L Ch R = 1,22109,246,246,246
BEGIN DESCRIPTION:
Mapping XS ef6670d5
END DESCRIPTION:
XS GIS Cut Line= 4
      2429399.20     13556281.27      2429438.99     13555846.10
      2429299.72     13555415.85      2429160.50     13555129.96
#Sta/Elev= 30
  4331.0  362.49  4467.8  358.77  4688.8  356.99  4766.0  355.38  4796.3  355.76
  4822.7  358.52  4842.7  361.39  4874.2  363.49  4897.6  363.30  4927.3  360.56
  4947.8  357.23  4954.3  354.36  4954.6  353.86  4958.1  353.86  4958.3  354.36
  5089.6  354.36  5095.0  358.00  5105.5  360.07  5116.0  361.15  5121.6  363.25
  5136.4  362.62  5147.5  361.52  5158.8  359.47  5179.1  359.51  5307.8  363.91
  5352.8  364.06  5358.4  364.95  5388.0  366.23  5432.5  367.10  5538.2  370.81
#Mann=6,-1,0
  4331.0    0.05       0  4822.7    0.04       0  4927.3     0.1       0
  4954.3    0.05       0  4958.3     0.1       0  5136.4    0.04       0
Bank Sta=4954.3,4958.3
Exp/Cntr=0.3,0.1

Type RM Length L Ch R = 1,21863,208,208,208
BEGIN DESCRIPTION:
Mapping XS c8e5f42a
END DESCRIPTION:
XS GIS Cut Line= 4
      2429468.85     13556176.82      2429610.59     13555634.70
      2429550.90     13555378.55      2429349.75     13555142.62
#Sta/Elev= 30
  4360.6  359.95  4366.4  360.14  4442.1  358.45  4497.3  357.76  4517.5  357.35
  4523.0  356.86  4528.2  357.07  4558.3  356.23  4589.9  356.09  4598.7  355.51
  4639.1  355.47  4672.6  354.73  4713.9  355.13  4751.9  354.71  4795.7  354.73
  4804.9  354.36  4805.2  353.86  4808.7  353.86  4808.9  354.36  4825.1  354.36
  4954.4  354.36  5105.5  354.36  5136.3  355.26  5204.6  355.45  5233.1  356.36
  5261.7  358.44  5296.8  360.09  5411.0  364.23  5452.7  364.74  5494.0  366.28
#Mann=7,-1,0
  4360.6    0.04       0  4497.3    0.05       0  4751.9    0.04       0
  4804.9    0.04       0  4808.9    0.04       0  4825.1    0.03       0
  4954.4    0.04       0
Bank Sta=4804.9,4808.9
Exp/Cntr=0.3,0.1

Type RM Length L Ch R = 1,21655,314,314,314
BEGIN DESCRIPTION:
Mapping XS 14f7d5eb
END DESCRIPTION:
XS GIS Cut Line= 5
      2429555.89     13556129.58      2429710.07     13555766.51
      2429787.17     13555617.30      2429729.97     13555371.09
      2429536.62     13555038.93
#Sta/Elev= 30
  4225.1  360.15  4327.9  358.74  4335.6  358.49  4349.6  356.41  4359.3  356.27
  4364.7  356.68  4369.5  358.91  4371.3  359.75  4388.4  356.38  4441.1  356.52
  4464.8  355.16  4493.9  355.63  4523.4  354.85  4593.9  355.19  4617.6  356.43
  4728.3  358.07  4766.9  357.94  4772.5  356.96  4797.7  357.31  4860.0  358.45
  4902.6  358.10  4907.7  357.08  4943.9  357.90  4955.5  356.94  5015.7  357.20
  5091.6  353.80  5091.8  353.30  5095.6  353.80  5267.2  357.55  5424.6  365.17
#Mann=5,-1,0
  4225.1    0.04       0  4369.5    0.03       0  4797.7    0.04       0
  5091.6    0.04       0  5095.6    0.04       0
Bank Sta=5091.6,5095.6
Exp/Cntr=0.3,0.1

Type RM Length L Ch R = 1,21341,325,325,325
BEGIN DESCRIPTION:
Mapping XS a3a8cf54
END DESCRIPTION:
XS GIS Cut Line= 3
      2430075.66     13555953.01      2430157.72     13555672.01
      2429889.57     13554974.30
#Sta/Elev= 30
  4335.0  357.08  4388.2  356.31  4421.6  354.00  4499.6  351.99  4527.2  352.55
  4532.5  351.91  4541.3  352.17  4560.7  353.76  4565.9  352.09  4599.4  355.88
  4604.6  353.70  4623.6  350.82  4656.7  350.48  4704.9  349.22  4720.9  349.46
  4784.3  348.18  4819.6  348.21  4828.1  347.70  4847.6  347.56  4847.9  347.06
  4851.4  347.06  4851.6  347.56  4958.9  348.65  4983.6  347.72  4999.5  347.82
  5038.2  349.89  5122.9  352.41  5309.3  356.11  5326.8  356.86  5375.2  358.47
#Mann=5,-1,0
  4335.0    0.04       0  4847.6    0.04       0  4851.6    0.04       0
  5309.3    0.05       0  5326.8    0.12       0
Bank Sta=4847.6,4851.6
Exp/Cntr=0.3,0.1

Type RM Length L Ch R = 1,21016,232,232,232
BEGIN DESCRIPTION:
Mapping XS 28d857e3
END DESCRIPTION:
XS GIS Cut Line= 3
      2430331.81     13556060.02      2430316.89     13555323.83
      2430075.64     13554940.81
#Sta/Elev= 30
  4264.4  358.14  4359.4  355.72  4449.5  354.14  4609.5  350.62  4709.5  349.20
  4779.5  349.16  4809.5  347.94  4850.9  347.37  4859.5  346.93  4959.6  346.77
  4979.6  345.49  5007.5  345.05  5007.7  344.55  5011.2  344.55  5011.5  345.05
  5051.9  346.07  5058.4  346.87  5067.2  347.32  5073.1  347.13  5088.4  348.18
  5140.1  349.77  5167.2  351.00  5197.8  351.49  5238.4  352.94  5370.9  356.31
  5386.2  357.38  5401.2  357.42  5408.5  357.89  5443.9  359.40  5453.4  359.44
#Mann=5,-1,0
  4264.4    0.04       0  5007.5    0.04       0  5011.5    0.04       0
  5238.4    0.05       0  5408.5    0.12       0
Bank Sta=5007.5,5011.5
Exp/Cntr=0.3,0.1

Type RM Length L Ch R = 1,20784,259,259,259
BEGIN DESCRIPTION:
Mapping XS 69c0efc6
END DESCRIPTION:
XS GIS Cut Line= 3
      2430560.61     13555985.34      2430548.18     13555303.94
      2430177.64     13554858.79
#Sta/Elev= 30
  4339.8  357.30  4640.2  349.68  4740.2  347.75  4814.2  347.15  4838.4  347.04
  4900.2  346.89  4918.3  345.93  5008.3  342.96  5008.5  342.46  5012.0  342.46
  5012.3  342.96  5023.9  343.15  5030.3  343.81  5036.8  343.66  5044.6  344.31
  5051.1  344.01  5079.7  346.18  5114.9  346.69  5157.8  347.95  5215.1  348.31
  5221.6  348.74  5305.9  350.42  5349.2  351.20  5444.0  354.60  5456.0  355.49
  5507.3  357.61  5534.1  359.16  5562.7  360.23  5577.0  361.41  5600.5  362.23
#Mann=8,-1,0
  4339.8    0.04       0  4814.2    0.05       0  4838.4    0.04       0
  5008.3    0.04       0  5012.3    0.04       0  5305.9    0.05       0
  5444.0    0.12       0  5507.3    0.05       0
Bank Sta=5008.3,5012.3
Exp/Cntr=0.3,0.1

Type RM Length L Ch R = 1,20525,405,405,405
BEGIN DESCRIPTION:
TRIB 3 TO YORKTOWN CREEK 38.0
END DESCRIPTION:
XS GIS Cut Line= 3
      2430974.98     13555824.95      2430775.00     13555225.00
      2430274.99     13554774.99
#Sta/Elev= 30
  4371.8  356.65  4424.5  353.54  4445.5  353.79  4508.8  350.78  4519.3  351.01
  4603.7  348.14  4614.2  348.70  4733.5  345.25  4772.3  344.55  4888.3  343.99
  4972.6  341.65  4991.7  341.61  4991.9  341.11  4995.4  341.11  4995.7  341.61
  5032.2  343.33  5152.6  345.86  5209.4  346.38  5259.5  348.28  5278.5  348.43
  5301.3  348.45  5329.7  349.51  5394.0  350.58  5506.8  353.85  5529.7  355.08
  5570.4  356.88  5613.0  359.62  5620.5  360.64  5641.4  361.14  5676.9  362.88
#Mann=8,-1,0
  4371.8    0.04       0  4733.5    0.05       0  4772.3    0.04       0
  4991.7    0.04       0  4995.7    0.04       0  5278.5    0.05       0
  5529.7    0.12       0  5641.4    0.05       0
Bank Sta=4991.7,4995.7
Exp/Cntr=0.3,0.1

Type RM Length L Ch R = 1,20120,224,224,224
BEGIN DESCRIPTION:
TRIB 3 TO YORKTOWN CREEK 37.0
END DESCRIPTION:
XS GIS Cut Line= 3
      2431125.00     13555875.00      2431075.00     13554975.00
      2430475.05     13554775.02
#Sta/Elev= 30
  4142.7  358.40  4192.8  356.22  4202.8  356.87  4244.4  355.13  4292.9  353.02
  4303.0  353.46  4344.2  351.48  4363.0  350.23  4373.1  350.95  4443.2  347.83
  4453.2  348.13  4603.4  344.23  4743.6  343.06  4783.7  341.93  4923.9  341.03
  4974.0  339.99  4992.0  338.88  4992.3  338.38  4995.8  338.38  4996.0  338.88
  5004.0  339.93  5014.0  340.19  5075.7  339.92  5123.0  341.59  5191.7  341.09
  5244.4  341.88  5360.3  344.87  5381.4  345.99  5434.1  346.59  5676.5  353.80
#Mann=6,-1,0
  4142.7    0.04       0  4244.4    0.05       0  4344.2    0.04       0
  4992.0    0.04       0  4996.0    0.04       0  5123.0    0.05       0
Bank Sta=4992,4996
Exp/Cntr=0.3,0.1

Type RM Length L Ch R = 1,19896,303,303,303
BEGIN DESCRIPTION:
Mapping XS de70d0ec
END DESCRIPTION:
XS GIS Cut Line= 3
      2431895.27     13555492.09      2431254.67     13554874.93
      2430599.22     13554627.84
#Sta/Elev= 30
  4058.9  351.07  4149.0  349.65  4219.7  346.76  4348.9  344.30  4424.7  343.32
  4502.7  341.05  4693.6  339.38  4813.7  339.27  4847.2  338.58  4847.5  338.08
  4851.0  338.08  4851.2  338.58  4863.4  339.28  4905.8  338.99  4920.0  339.57
  4926.9  338.97  4963.3  338.58  4980.1  339.06  5048.5  338.59  5078.7  339.01
  5103.6  340.31  5164.0  339.82  5196.9  340.65  5334.5  343.26  5444.7  346.20
  5450.4  346.77  5524.6  347.87  5529.9  347.39  5535.9  347.99  5648.9  350.54
#Mann=5,-1,0
  4058.9    0.05       0  4348.9    0.04       0  4847.2    0.04       0
  4851.2    0.04       0  5196.9    0.05       0
Bank Sta=4847.2,4851.2
Exp/Cntr=0.3,0.1

Type RM Length L Ch R = 1,19593,540,540,540
BEGIN DESCRIPTION:
TRIB 3 TO YORKTOWN CREEK 36.0
END DESCRIPTION:
XS GIS Cut Line= 3
      2432025.02     13555325.02      2431425.00     13554725.00
      2430675.00     13553825.00
#Sta/Elev= 30
  4071.8  352.50  4156.7  349.76  4354.7  345.32  4482.0  340.74  4552.7  339.45
  4722.4  337.94  4736.5  337.29  4849.7  337.65  4863.8  337.09  4948.3  337.94
  4956.2  337.32  4991.3  336.97  5040.8  337.35  5074.6  336.70  5074.8  336.20
  5078.3  336.20  5078.6  336.70  5090.2  337.21  5275.1  338.62  5367.5  340.46
  5474.2  340.11  5587.5  343.11  5630.4  343.01  5694.2  344.61  5708.5  344.18
  5772.3  346.57  5807.5  349.26  5843.9  349.41  5928.5  352.22  6091.9  359.36
#Mann=3,-1,0
  4071.8    0.04       0  5074.6    0.04       0  5078.6    0.04       0
Bank Sta=5074.6,5078.6
Exp/Cntr=0.3,0.1

Type RM Length L Ch R = 1,19053,514,514,514
BEGIN DESCRIPTION:
TRIB 3 TO YORKTOWN CREEK 35.0
END DESCRIPTION:
XS GIS Cut Line= 3
      2432325.03     13554975.03      2431725.00     13554375.00
      2431125.00     13553775.00
#Sta/Elev= 30
  4005.8  351.63  4063.6  350.06  4147.3  348.23  4218.0  345.17  4359.4  341.06
  4486.7  338.47  4515.0  339.25  4559.4  337.32  4656.4  335.47  4755.4  334.65
  4826.1  334.45  4917.5  335.07  4967.5  333.97  4979.7  333.04  4979.9  332.54
  4983.4  332.54  4983.7  333.04  5024.1  334.97  5094.8  335.60  5165.5  337.75
  5188.8  337.53  5207.9  338.11  5306.9  338.17  5333.4  339.08  5377.6  339.75
  5405.9  339.54  5427.4  340.18  5476.6  341.84  5547.3  343.28  5702.9  349.19
#Mann=9,-1,0
  4005.8    0.05       0  4063.6    0.04       0  4559.4    0.05       0
  4917.5    0.03       0  4979.7    0.03       0  4983.7    0.03       0
  5188.8    0.04       0  5333.4    0.05       0  5427.4    0.04       0
Bank Sta=4979.7,4983.7
Exp/Cntr=0.3,0.1

Type RM Length L Ch R = 1,18539,559,559,559
BEGIN DESCRIPTION:
TRIB 3 TO YORKTOWN CREEK 34.0
END DESCRIPTION:
XS GIS Cut Line= 3
      2432574.99     13554674.99      2432025.00     13554075.00
      2431424.97     13553474.97
#Sta/Elev= 30
  4009.3  351.59  4250.1  342.07  4401.5  337.96  4525.7  334.95  4646.6  333.07
  4724.3  333.48  4759.4  332.93  4830.1  333.61  4851.5  333.76  4879.8  337.07
  4908.1  339.15  4929.3  338.69  4950.5  335.52  4964.6  332.69  5075.8  332.62
  5076.0  332.12  5079.5  332.12  5079.8  332.62  5091.9  334.02  5106.1  336.70
  5120.2  338.44  5141.4  337.96  5176.8  334.96  5190.9  335.45  5233.3  334.68
  5275.8  336.34  5327.5  337.11  5374.8  337.67  5445.5  339.41  5671.8  345.82
#Mann=6,-1,0
  4009.3    0.04       0  4401.5    0.05       0  4830.1    0.03       0
  5075.8    0.03       0  5079.8    0.03       0  5327.5    0.04       0
Bank Sta=5075.8,5079.8
Exp/Cntr=0.3,0.1

Type RM Length L Ch R = 1,17980,479,479,479
BEGIN DESCRIPTION:
TRIB 3 TO YORKTOWN CREEK 33.0
END DESCRIPTION:
XS GIS Cut Line= 3
      2432674.99     13554324.99      2432275.00     13553725.00
      2431675.02     13553425.01
#Sta/Elev= 30
  4279.5  341.42  4374.1  338.60  4473.3  336.20  4509.3  335.87  4539.4  334.99
  4626.5  333.46  4683.6  332.64  4725.7  332.64  4812.8  331.88  4878.9  330.79
  4899.9  331.43  4921.0  331.57  4936.0  331.22  4957.0  331.86  4995.6  329.51
  4995.8  329.01  4999.3  329.01  4999.6  329.51  5014.6  329.85  5031.3  331.39
  5036.9  332.31  5053.7  332.58  5076.1  332.48  5104.0  331.69  5157.1  332.65
  5215.8  332.46  5260.5  331.87  5367.0  333.13  5461.8  334.53  5671.4  340.11
#Mann=4,-1,0
  4279.5    0.05       0  4995.6    0.05       0  4999.6    0.05       0
  5367.0    0.04       0
Bank Sta=4995.6,4999.6
Exp/Cntr=0.3,0.1

Type RM Length L Ch R = 1,17501,556,556,556
BEGIN DESCRIPTION:
TRIB 3 TO YORKTOWN CREEK 32.0
END DESCRIPTION:
XS GIS Cut Line= 3
      2433174.99     13553974.99      2432575.00     13553375.00
      2431674.95     13553274.99
#Sta/Elev= 30
  4102.9  341.35  4201.9  337.39  4272.6  335.65  4414.0  333.18  4531.4  332.04
  4696.9  330.25  4881.6  329.32  4971.5  328.87  4991.7  328.25  5001.7  327.16
  5020.8  327.43  5029.9  327.01  5030.2  326.51  5033.7  326.51  5033.9  327.01
  5042.0  327.09  5052.0  328.57  5072.2  328.42  5122.5  329.29  5203.0  329.04
  5253.3  329.40  5323.7  330.77  5343.8  330.61  5504.8  332.93  5615.5  334.99
  5685.9  336.80  5726.2  337.19  5796.6  338.90  5826.8  340.12  5857.0  340.59
#Mann=6,-1,0
  4102.9    0.04       0  4531.4    0.05       0  4881.6    0.12       0
  5020.8    0.04       0  5029.9    0.05       0  5033.9    0.04       0
Bank Sta=5029.9,5033.9
Exp/Cntr=0.3,0.1

Type RM Length L Ch R = 1,16945,557,557,557
BEGIN DESCRIPTION:
TRIB 3 TO YORKTOWN CREEK 31.0
END DESCRIPTION:
XS GIS Cut Line= 3
      2433475.03     13553625.03      2432875.00     13553025.00
      2432325.01     13552425.01
#Sta/Elev= 30
  4012.3  339.59  4139.6  336.35  4167.9  334.85  4182.1  334.94  4196.2  334.16
  4210.3  334.72  4252.8  332.35  4295.2  331.81  4309.3  330.95  4365.9  329.51
  4467.0  328.99  4493.2  328.19  4595.0  327.17  4691.2  326.46  4747.7  327.07
  4967.0  326.92  4981.4  326.73  4993.4  325.50  4993.7  325.00  4997.6  325.00
  4997.9  325.50  5002.4  326.28  5016.6  326.82  5101.9  327.30  5121.6  327.69
  5186.5  328.18  5193.5  328.70  5264.5  329.61  5429.5  333.08  5674.8  338.95
#Mann=9,-1,0
  4012.3    0.05       0  4467.0    0.04       0  4595.0    0.05       0
  4967.0    0.04       0  4993.4    0.04       0  4997.9    0.04       0
  5101.9    0.03       0  5121.6    0.04       0  5429.5    0.03       0
Bank Sta=4993.4,4997.9
Exp/Cntr=0.3,0.1

Type RM Length L Ch R = 1,16388,498,498,498
BEGIN DESCRIPTION:
TRIB 3 TO YORKTOWN CREEK 30.0
END DESCRIPTION:
XS GIS Cut Line= 3
      2433775.01     13553525.02      2433075.00     13552625.00
      2432475.02     13552025.02
#Sta/Elev= 30
  4106.9  341.37  4220.9  337.40  4358.9  334.30  4452.9  332.82  4649.0  327.68
  5024.0  324.03  5024.3  323.53  5028.7  324.03  5055.8  325.33  5080.0  325.47
  5119.5  325.30  5140.3  326.58  5146.7  328.89  5161.1  330.10  5196.4  329.78
  5204.6  330.81  5210.9  329.94  5219.0  330.73  5225.4  329.53  5233.5  330.37
  5239.9  328.93  5243.9  330.00  5289.5  330.57  5332.0  326.42  5347.1  326.34
  5529.9  329.01  5727.9  335.08  5789.8  336.07  5864.8  338.02  6095.6  346.37
#Mann=10,-1,0
  4106.9    0.05       0  4358.9    0.04       0  4452.9    0.05       0
  5024.0    0.05       0  5028.7    0.05       0  5055.8    0.12       0
  5080.0    0.05       0  5347.1    0.04       0  5789.8    0.03       0
  5864.8    0.04       0
Bank Sta=5024,5028.7
Exp/Cntr=0.3,0.1

Type RM Length L Ch R = 1,15890,453,453,453
BEGIN DESCRIPTION:
TRIB 3 TO YORKTOWN CREEK 29.0
END DESCRIPTION:
XS GIS Cut Line= 3
      2434124.99     13553174.99      2433375.00     13552375.00
      2432574.99     13551674.99
#Sta/Elev= 30
  3903.4  335.04  3960.0  334.52  4052.1  332.38  4158.1  330.63  4193.3  330.62
  4278.3  328.85  4883.0  323.29  4936.7  324.16  4971.9  323.30  4992.9  320.69
  4994.1  320.00  4994.4  319.50  4998.6  319.50  4999.0  320.00  5028.0  320.52
  5042.2  321.84  5078.3  323.52  5106.3  324.02  5177.0  323.54  5212.6  324.10
  5311.8  326.49  5326.0  327.33  5389.6  327.96  5503.5  331.47  5545.2  332.14
  5613.0  334.54  5644.9  336.34  5744.1  339.41  5856.7  344.01  6063.0  351.07
#Mann=8,-1,0
  3903.4    0.04       0  3960.0    0.05       0  4883.0   0.013       0
  4936.7    0.05       0  4994.1    0.05       0  4999.0    0.05       0
  5613.0   0.013       0  5856.7    0.04       0
Bank Sta=4994.1,4999
Exp/Cntr=0.3,0.1

Type RM Length L Ch R = 1,15437,419,419,419
BEGIN DESCRIPTION:
TRIB 3 TO YORKTOWN CREEK 28.0
END DESCRIPTION:
XS GIS Cut Line= 3
      2434324.98     13552774.98      2433525.00     13551975.00
      2432925.05     13551725.02
#Sta/Elev= 30
  3830.3  341.55  3858.6  341.29  3886.8  338.70  3901.0  335.94  3945.7  332.80
  4084.8  328.94  4113.1  328.99  4127.3  330.04  4141.4  329.52  4156.4  327.59
  4169.7  326.43  4183.8  326.20  4252.1  326.35  4353.5  325.82  4509.1  322.86
  4650.5  323.39  4735.4  321.86  4905.1  323.12  4955.6  320.40  4980.8  319.10
  4981.2  318.60  4985.4  318.60  4985.8  319.10  4994.1  319.12  5015.8  321.95
  5037.5  323.22  5135.5  323.70  5330.0  327.88  5390.1  330.97  5611.6  340.03
#Mann=7,-1,0
  3830.3    0.03       0  3945.7    0.04       0  4156.4    0.05       0
  4252.1    0.03       0  4955.6    0.05       0  4980.8    0.05       0
  4985.8    0.05       0
Bank Sta=4980.8,4985.8
Exp/Cntr=0.3,0.1

Type RM Length L Ch R = 1,15018,474,474,474
BEGIN DESCRIPTION:
TRIB 3 TO YORKTOWN CREEK 27.0
END DESCRIPTION:
XS GIS Cut Line= 3
      2434325.01     13552625.01      2433825.00     13551775.00
      2433224.97     13551324.98
#Sta/Elev= 30
  4087.3  341.54  4110.5  340.41  4122.4  334.94  4132.3  333.62  4175.8  331.98
  4202.7  330.79  4233.8  330.43  4261.3  326.83  4505.0  325.98  4532.5  325.42
  4569.7  323.11  4612.6  322.96  4702.2  320.54  4833.7  320.97  4878.8  320.39
  4950.1  320.72  4979.8  319.94  5028.5  321.10  5038.4  319.90  5044.2  321.19
  5057.3  319.16  5057.7  318.66  5062.3  319.16  5063.7  319.79  5065.6  320.64
  5187.5  321.27  5307.8  321.64  5480.8  322.46  5601.6  324.35  5823.5  331.25
#Mann=11,-1,0
  4087.3    0.03       0  4175.8    0.04       0  4202.7    0.03       0
  4833.7    0.05       0  4878.8    0.12       0  4950.1    0.05       0
  5057.3    0.05       0  5062.3    0.05       0  5063.7    0.12       0
  5187.5   0.013       0  5307.8    0.05       0
Bank Sta=5057.3,5062.3
Exp/Cntr=0.3,0.1

Type RM Length L Ch R = 1,14544,496,496,496
BEGIN DESCRIPTION:
TRIB 3 TO YORKTOWN CREEK 26.0
END DESCRIPTION:
XS GIS Cut Line= 3
      2434325.00     13552475.02      2434225.00     13551575.00
      2433024.96     13551074.98
#Sta/Elev= 30
  4184.4  330.21  4214.6  326.77  4476.2  325.45  4486.3  323.78  4506.4  322.23
  4586.9  320.80  4617.1  319.47  4748.9  318.74  4834.2  318.47  4949.1  319.00
  4959.2  318.35  5016.4  319.84  5087.4  318.88  5122.5  319.66  5125.9  318.33
  5126.3  317.83  5130.9  318.33  5241.6  318.65  5258.4  319.26  5295.9  318.90
  5359.2  318.73  5430.4  319.61  5611.8  321.17  5717.1  321.30  5761.6  322.10
  5807.7  321.36  5915.4  324.15  6093.0  328.55  6296.3  333.65  6390.0  336.44
#Mann=13,-1,0
  4184.4    0.03       0  4748.9    0.05       0  4834.2    0.12       0
  5016.4    0.05       0  5125.9    0.05       0  5130.9    0.05       0
  5295.9    0.12       0  5430.4    0.05       0  5611.8   0.013       0
  5717.1    0.05       0  5915.4    0.03       0  6093.0    0.05       0
  6296.3    0.03       0
Bank Sta=5125.9,5130.9
Exp/Cntr=0.3,0.1

Type RM Length L Ch R = 1,14048,467,467,467
BEGIN DESCRIPTION:
TRIB 3 TO YORKTOWN CREEK 25.0
END DESCRIPTION:
XS GIS Cut Line= 3
      2435124.98     13552374.97      2434675.00     13551475.00
      2434125.02     13551025.02
#Sta/Elev= 30
  3958.3  329.16  4026.4  326.81  4030.2  326.71  4092.4  325.28  4123.2  323.84
  4173.5  323.04  4195.8  321.80  4204.2  322.30  4212.6  321.38  4262.9  320.00
  4310.0  319.33  4319.4  319.29  4383.1  318.98  4427.8  317.94  4480.9  318.30
  4525.3  317.77  4584.4  316.94  4665.4  317.11  4749.3  315.94  4928.2  316.33
  5016.4  315.34  5018.7  315.09  5019.1  314.59  5023.3  314.59  5023.7  315.09
  5255.9  317.72  5362.9  321.24  5480.3  323.72  5561.0  325.48  5675.1  326.20
#Mann=10,-1,0
  3958.3    0.05       0  4026.4    0.04       0  4030.2    0.05       0
  4310.0    0.04       0  4319.4    0.05       0  4525.3    0.04       0
  5016.4    0.05       0  5018.7    0.04       0  5023.7    0.05       0
  5480.3    0.04       0
Bank Sta=5018.7,5023.7
Exp/Cntr=0.3,0.1

Type RM Length L Ch R = 1,13581,505,505,505
BEGIN DESCRIPTION:
TRIB 3 TO YORKTOWN CREEK 24.0
END DESCRIPTION:
XS GIS Cut Line= 3
      2435825.03     13552025.03      2435025.00     13551125.00
      2434274.96     13551075.00
#Sta/Elev= 30
  3748.5  327.52  3769.9  327.02  3790.8  327.34  3855.2  325.22  3861.8  324.47
  3876.1  324.50  3882.8  323.45  3911.2  321.54  3925.4  321.63  3947.1  320.74
  4081.8  318.01  4102.7  318.05  4201.6  316.17  4265.7  315.10  4286.6  315.40
  4308.4  314.73  4378.6  315.98  4506.6  314.41  4777.4  314.19  5000.3  312.66
  5000.6  312.16  5005.0  312.16  5005.4  312.66  5062.9  313.59  5133.1  313.37
  5323.5  315.17  5349.3  315.84  5443.8  317.38  5644.2  324.66  5704.4  325.72
#Mann=6,-1,0
  3748.5    0.05       0  4201.6    0.04       0  4777.4    0.05       0
  5000.3    0.05       0  5005.4    0.05       0  5349.3    0.04       0
Bank Sta=5000.3,5005.4
Exp/Cntr=0.3,0.1

Type RM Length L Ch R = 1,13076,440,440,440
BEGIN DESCRIPTION:
TRIB 3 TO YORKTOWN CREEK 23.0
END DESCRIPTION:
XS GIS Cut Line= 3
      2436074.97     13551674.96      2435325.00     13550775.00
      2434824.98     13549874.96
#Sta/Elev= 30
  3897.1  321.90  3996.6  317.64  4017.5  314.24  4025.3  316.22  4031.8  312.89
  4039.6  314.16  4046.1  312.56  4060.4  316.14  4066.9  314.31  4081.2  316.39
  4089.1  319.21  4109.9  320.13  4181.5  313.05  4337.7  311.98  4344.2  309.67
  4352.0  309.30  4450.9  309.31  4458.2  311.38  4461.0  311.31  4508.2  314.53
  4607.1  311.10  5091.5  311.71  5423.2  309.23  5480.4  310.44  5553.6  309.00
  5557.9  307.48  5558.3  306.98  5563.0  307.48  5591.4  309.83  6098.2  324.52
#Mann=5,-1,0
  3897.1    0.05       0  4458.2   0.013       0  4461.0    0.04       0
  5557.9    0.04       0  5563.0    0.04       0
Bank Sta=5557.9,5563
Exp/Cntr=0.3,0.1

Type RM Length L Ch R = 1,12636,565,565,565
BEGIN DESCRIPTION:
TRIB 3 TO YORKTOWN CREEK 22.0
END DESCRIPTION:
XS GIS Cut Line= 3
      2436625.00     13551575.00      2435425.00     13550375.00
      2434924.98     13549774.98
#Sta/Elev= 30
  3649.0  323.37  3886.2  318.98  4070.2  315.97  4158.1  313.67  4373.8  311.20
  4380.0  311.29  4455.1  309.86  4735.3  308.10  4735.7  307.60  4740.5  308.10
  5176.3  309.78  5310.7  309.19  5388.4  310.05  5437.8  309.15  5488.6  309.99
  5495.1  311.70  5509.4  309.67  5515.9  310.70  5523.7  309.81  5530.2  310.81
  5538.1  309.64  5544.6  311.01  5552.4  310.22  5558.9  310.97  5566.7  309.81
  5573.2  310.79  5587.5  308.90  5722.9  311.92  5920.8  320.98  6127.1  326.44
#Mann=7,-1,0
  3649.0   0.035       0  3886.2    0.05       0  4070.2    0.04       0
  4373.8   0.013       0  4380.0    0.04       0  4735.3    0.04       0
  4740.5    0.04       0
Bank Sta=4735.3,4740.5
Exp/Cntr=0.3,0.1

Type RM Length L Ch R = 1,12071,397,397,397
BEGIN DESCRIPTION:
TRIB 3 TO YORKTOWN CREEK 21.0
END DESCRIPTION:
XS GIS Cut Line= 3
      2436825.03     13551225.03      2435625.00     13550025.00
      2435075.02     13549675.01
#Sta/Elev= 30
  3974.8  322.52  4088.0  320.16  4175.6  319.82  4314.3  314.58  4526.4  310.42
  4690.4  308.66  4825.6  307.82  4905.5  306.97  4960.8  306.62  4990.2  306.15
  4990.7  305.65  4995.5  305.65  4996.0  306.15  5049.0  307.25  5096.0  307.14
  5192.5  307.26  5231.2  307.20  5360.8  307.47  5502.2  308.74  5674.9  308.17
  5707.5  306.66  5731.2  306.47  5773.5  307.91  5825.1  308.05  5991.9  311.85
  6063.1  316.42  6179.9  319.75  6222.2  321.54  6279.8  325.25  6323.8  326.25
#Mann=12,-1,0
  3974.8   0.035       0  4175.6    0.04       0  4690.4   0.013       0
  4825.6    0.04       0  4905.5   0.013       0  4960.8    0.04       0
  4990.2    0.04       0  4996.0    0.04       0  5049.0    0.05       0
  5096.0    0.04       0  5192.5    0.05       0  5231.2    0.04       0
Bank Sta=4990.2,4996
Exp/Cntr=0.3,0.1

Type RM Length L Ch R = 1,11674,399,399,399
BEGIN DESCRIPTION:
TRIB 3 TO YORKTOWN CREEK 20.0
END DESCRIPTION:
XS GIS Cut Line= 3
      2436825.00     13550825.00      2435825.00     13549625.00
      2435524.97     13549374.98
#Sta/Elev= 30
  4139.0  316.03  4437.7  309.93  4501.5  309.66  4594.0  307.96  4672.1  305.72
  4863.3  306.62  4894.4  306.58  4920.0  305.28  4976.7  305.36  4991.0  304.40
  5016.7  303.99  5017.2  303.49  5022.5  303.99  5076.2  304.26  5182.3  306.37
  5239.6  306.28  5253.9  306.39  5260.4  307.14  5288.4  307.08  5352.8  307.69
  5431.0  306.59  5492.7  306.77  5650.9  306.19  5708.2  304.94  5743.4  305.34
  5800.6  306.93  5850.1  307.45  5921.7  310.07  6027.1  312.63  6091.6  315.80
#Mann=7,-1,0
  4139.0    0.04       0  4863.3    0.05       0  4894.4    0.04       0
  5016.7    0.04       0  5022.5    0.04       0  5288.4   0.013       0
  5492.7    0.04       0
Bank Sta=5016.7,5022.5
Exp/Cntr=0.3,0.1

Type RM Length L Ch R = 1,11275,867,867,867
BEGIN DESCRIPTION:
TRIB 3 TO YORKTOWN CREEK 19.0
END DESCRIPTION:
XS GIS Cut Line= 3
      2437075.01     13550825.01      2436175.00     13549325.00
      2435575.02     13548975.01
#Sta/Elev= 30
  3941.1  317.24  4070.1  315.36  4166.6  312.94  4384.3  309.88  4399.8  309.08
  4421.2  309.42  4473.7  307.51  4617.5  304.99  4722.5  304.53  4808.0  305.13
  4839.1  304.25  4897.4  304.89  5011.1  302.90  5011.6  302.40  5016.9  302.90
  5025.7  303.86  5049.0  303.38  5142.3  304.68  5391.1  303.69  5566.0  304.88
  5693.3  303.54  5771.4  305.08  5829.3  305.17  5923.2  307.91  5928.9  307.48
  5950.0  307.49  6136.5  310.86  6275.5  316.33  6312.7  316.38  6385.0  318.75
#Mann=6,-1,0
  3941.1   0.035       0  4070.1    0.04       0  5011.1    0.04       0
  5016.9    0.04       0  5928.9   0.013       0  5950.0    0.04       0
Bank Sta=5011.1,5016.9
Exp/Cntr=0.3,0.1

Type RM Length L Ch R = 1,10408,605,605,605
BEGIN DESCRIPTION:
Mapping XS ad4f4a38
END DESCRIPTION:
XS GIS Cut Line= 4
      2437537.66     13550702.19      2437240.82     13549641.24
      2436666.07     13549128.34      2435764.01     13548788.14
#Sta/Elev= 30
  3209.0  314.33  3343.7  312.12  3398.2  311.14  3940.4  302.27  4110.8  301.82
  4291.6  301.08  4677.8  302.21  4708.5  302.33  4730.2  305.43  4751.1  306.55
  4783.8  302.50  4793.7  302.41  4804.2  300.25  4804.7  299.75  4811.6  300.25
  4814.6  301.48  4822.2  300.46  4843.1  302.41  4864.8  302.03  4871.5  303.94
  4893.2  304.50  4914.1  306.99  4965.2  302.96  5191.8  301.80  5295.8  302.40
  5461.7  303.74  5637.8  305.86  5643.2  307.12  5764.0  309.38  6045.1  315.30
#Mann=14,-1,0
  3209.0    0.04       0  3343.7    0.05       0  3398.2    0.04       0
  4110.8    0.05       0  4291.6    0.04       0  4677.8    0.05       0
  4783.8    0.04       0  4804.2    0.05       0  4811.6    0.04       0
  4965.2    0.05       0  5191.8    0.04       0  5295.8    0.05       0
  5461.7   0.013       0  5764.0    0.05       0
Bank Sta=4804.2,4811.6
Exp/Cntr=0.3,0.1

Type RM Length L Ch R = 1,9803,922,922,922
BEGIN DESCRIPTION:
Mapping XS d52185ca
END DESCRIPTION:
XS GIS Cut Line= 3
      2437719.94     13550556.31      2437397.00     13549016.55
      2435803.28     13548696.98
#Sta/Elev= 30
  3147.8  310.62  3517.0  303.73  3772.4  300.76  4495.8  299.72  4510.4  300.22
  4528.5  299.18  4549.0  300.53  4586.1  298.21  4586.6  297.71  4593.5  298.21
  4607.1  300.18  4639.8  300.49  4657.0  302.13  4712.4  302.94  4858.5  301.78
  4947.5  301.35  4998.5  298.31  5066.7  300.43  5166.4  301.30  5254.7  301.57
  5266.1  301.64  5365.9  302.12  5457.4  299.97  5488.0  302.16  5515.4  302.57
  5783.8  303.54  6059.2  307.84  6089.8  309.94  6284.0  313.25  6346.5  315.10
#Mann=13,-1,0
  3147.8    0.04       0  4495.8    0.05       0  4510.4   0.013       0
  4586.1    0.05       0  4593.5   0.013       0  4639.8    0.05       0
  4858.5    0.12       0  5066.7    0.05       0  5166.4   0.013       0
  5254.7    0.05       0  5266.1    0.12       0  5365.9    0.05       0
  6284.0    0.04       0
Bank Sta=4586.1,4593.5
Exp/Cntr=0.3,0.1

Type RM Length L Ch R = 1,8881,514,514,514
BEGIN DESCRIPTION:
Mapping XS dbbf72f6
END DESCRIPTION:
XS GIS Cut Line= 3
      2437865.78     13550342.80      2438048.07     13549113.65
      2437428.27     13547400.09
#Sta/Elev= 30
  3502.5  305.17  3542.4  304.64  3759.7  302.07  3765.8  302.00  4283.5  297.93
  4517.6  297.87  4602.2  296.86  4616.8  298.04  4694.2  298.34  4723.5  300.31
  4769.5  297.26  4836.3  297.95  4948.1  298.82  4973.5  297.67  4994.0  292.92
  4994.5  292.42  5003.5  292.92  5030.4  294.70  5083.9  299.97  5272.7  302.31
  5392.3  303.39  5456.1  306.23  5503.9  305.51  5559.9  308.23  5590.5  307.39
  5924.0  316.56  5976.5  316.63  6236.2  322.36  6506.3  327.05  6567.3  328.65
#Mann=15,-1,0
  3502.5    0.05       0  3542.4    0.04       0  3759.7    0.05       0
  3765.8    0.04       0  4283.5    0.05       0  4517.6   0.013       0
  4616.8    0.05       0  4836.3    0.12       0  4994.0    0.05       0
  5003.5    0.12       0  5030.4    0.05       0  5272.7    0.04       0
  5976.5    0.03       0  6236.2    0.04       0  6506.3    0.03       0
Bank Sta=4994,5003.5
Exp/Cntr=0.3,0.1

Type RM Length L Ch R = 1,8367,339,339,339
BEGIN DESCRIPTION:
Mapping XS 5121e03d
END DESCRIPTION:
XS GIS Cut Line= 3
      2438037.65     13550665.77      2438391.82     13548728.23
      2438584.53     13547275.10
#Sta/Elev= 30
  3042.0  311.88  3098.0  310.82  3187.3  308.52  3226.4  308.87  3286.9  305.17
  3534.6  301.68  3933.7  298.10  4161.0  296.67  4225.0  298.65  4302.4  296.77
  4323.7  297.07  4364.3  302.15  4389.8  297.72  4412.3  297.12  4740.5  296.33
  4782.6  297.10  4811.6  300.91  4889.1  296.39  4947.4  296.81  5020.2  293.60
  5020.7  293.10  5029.8  293.60  5080.7  297.60  5179.7  297.73  5599.4  302.04
  5902.6  304.55  6033.7  307.60  6154.8  307.00  6212.6  309.93  6477.5  313.29
#Mann=13,-1,0
  3042.0    0.04       0  3098.0   0.013       0  3187.3    0.04       0
  3286.9    0.05       0  3534.6    0.04       0  3933.7    0.05       0
  4302.4   0.013       0  4412.3    0.05       0  5020.2    0.05       0
  5029.8    0.05       0  5080.7   0.013       0  5179.7    0.05       0
  5599.4    0.04       0
Bank Sta=5020.2,5029.8
Exp/Cntr=0.3,0.1

Type RM Length L Ch R = 1,8028,331,331,331
BEGIN DESCRIPTION:
Mapping XS 30945a94
END DESCRIPTION:
XS GIS Cut Line= 3
      2438339.74     13550514.68      2438667.86     13548816.77
      2438907.25     13547599.00
#Sta/Elev= 30
  3271.4  313.01  3326.3  312.62  3378.1  310.99  3444.2  310.83  3474.8  309.05
  3546.1  307.54  3576.6  305.91  3694.1  303.22  4096.1  296.25  4802.8  295.86
  4870.1  295.04  4900.7  295.63  4951.6  293.90  4992.3  294.07  4999.1  291.77
  5004.9  291.14  5005.4  290.64  5014.5  291.14  5014.8  291.91  5033.1  294.34
  5061.1  295.84  5169.0  294.99  5528.8  298.14  5688.1  300.36  5746.5  302.86
  5824.0  303.50  6093.0  306.25  6150.7  308.41  6207.2  308.28  6241.8  309.36
#Mann=5,-1,0
  3271.4    0.04       0  4802.8    0.05       0  5004.9    0.05       0
  5014.5    0.05       0  5824.0    0.04       0
Bank Sta=5004.9,5014.5
Exp/Cntr=0.3,0.1

Type RM Length L Ch R = 1,7697,529,529,529
BEGIN DESCRIPTION:
Mapping XS 53c4e671
END DESCRIPTION:
XS GIS Cut Line= 3
      2438824.12     13549983.41      2438969.95     13548868.85
      2439001.20     13547842.79
#Sta/Elev= 30
  3920.6  304.91  4029.9  302.25  4070.3  301.99  4196.8  298.18  4201.8  298.73
  4251.8  297.03  4322.4  296.05  4453.5  295.21  4507.2  295.55  4675.4  293.62
  4766.2  294.97  4848.1  294.70  4927.5  294.72  4957.8  293.90  4970.5  293.47
  4993.3  291.15  4993.8  290.65  5002.4  290.65  5002.9  291.15  5050.0  292.47
  5068.5  294.05  5088.5  294.49  5138.6  295.13  5218.6  293.70  5495.1  297.53
  5698.6  299.43  5718.8  299.07  5798.9  301.33  5835.5  301.52  6071.2  304.84
#Mann=7,-1,0
  3920.6    0.04       0  4848.1    0.05       0  4957.8    0.04       0
  4993.3    0.04       0  5002.9    0.04       0  5495.1    0.05       0
  5835.5    0.04       0
Bank Sta=4993.3,5002.9
Exp/Cntr=0.3,0.1

Type RM Length L Ch R = 1,7168,498,498,498
BEGIN DESCRIPTION:
TRIB 3 TO YORKTOWN CREEK 11.0
END DESCRIPTION:
XS GIS Cut Line= 3
      2439175.00     13550075.00      2439475.00     13548875.00
      2439075.01     13547675.04
#Sta/Elev= 30
  3758.5  318.14  3810.0  315.59  3841.0  314.73  3859.0  313.06  3864.2  313.59
  3882.2  311.43  3982.7  306.79  4147.6  300.92  4214.3  299.47  4304.8  297.83
  4552.2  295.38  4565.1  294.77  4624.4  294.64  4665.6  293.49  4830.5  292.63
  4871.7  292.97  4892.1  292.42  4956.2  290.70  5000.9  289.53  5001.4  289.03
  5010.6  289.03  5011.1  289.53  5111.4  292.17  5259.0  292.07  5415.1  293.85
  5480.3  295.83  5680.6  297.64  5798.1  299.30  6049.5  303.26  6260.3  307.86
#Mann=8,-1,0
  3758.5    0.05       0  4214.3    0.04       0  4892.1    0.05       0
  4956.2    0.04       0  5000.9    0.04       0  5011.1    0.04       0
  5415.1    0.05       0  5798.1    0.04       0
Bank Sta=5000.9,5011.1
Exp/Cntr=0.3,0.1

Type RM Length L Ch R = 1,6670,762,762,762
BEGIN DESCRIPTION:
TRIB 3 TO YORKTOWN CREEK 10.0
END DESCRIPTION:
XS GIS Cut Line= 3
      2439825.00     13549574.98      2439925.00     13548825.00
      2439325.00     13547725.01
#Sta/Elev= 30
  4248.9  303.80  4309.4  302.52  4441.8  297.54  4588.1  293.43  4712.9  291.87
  4904.6  290.39  4945.0  289.16  4963.9  287.81  4968.9  288.04  4980.1  287.36
  4980.6  286.86  4990.0  286.86  4990.5  287.36  5013.6  289.07  5051.1  290.26
  5117.0  289.14  5166.4  289.53  5198.7  290.53  5433.1  292.27  5483.9  292.83
  5492.9  293.52  5558.4  293.06  5623.9  293.70  5654.8  295.16  5699.9  294.81
  5755.2  296.12  5999.8  300.55  6103.3  303.02  6184.9  305.74  6258.5  306.83
#Mann=5,-1,0
  4248.9    0.04       0  4980.1    0.04       0  4990.5    0.04       0
  5433.1    0.05       0  5755.2    0.04       0
Bank Sta=4980.1,4990.5
Exp/Cntr=0.3,0.1

Type RM Length L Ch R = 1,5908,548,548,548
BEGIN DESCRIPTION:
Mapping XS feca892f
END DESCRIPTION:
XS GIS Cut Line= 3
      2440272.04     13549629.22      2440495.99     13548707.40
      2440116.13     13547859.21
#Sta/Elev= 30
  4008.7  299.65  4064.5  298.90  4087.5  299.36  4124.1  299.02  4146.8  297.02
  4177.7  295.97  4321.8  294.98  4371.5  294.11  4463.4  295.31  4733.4  289.93
  4927.9  288.41  4933.0  288.95  5014.8  285.97  5015.3  283.86  5015.8  283.36
  5025.4  283.36  5025.9  283.86  5043.8  287.02  5067.0  287.91  5095.6  288.46
  5113.3  289.43  5118.8  288.96  5158.2  288.79  5162.2  288.77  5268.9  288.83
  5361.7  289.69  5436.7  291.32  5511.8  291.49  5656.4  293.98  5886.7  296.81
#Mann=6,-1,0
  4008.7    0.05       0  4371.5    0.12       0  5015.3    0.05       0
  5025.9    0.12       0  5158.2    0.05       0  5162.2   0.035       0
Bank Sta=5015.3,5025.9
Exp/Cntr=0.3,0.1

Type RM Length L Ch R = 1,5360,675,675,675
BEGIN DESCRIPTION:
Mapping XS c81e085a
END DESCRIPTION:
XS GIS Cut Line= 3
      2441120.99     13549577.22      2440985.57     13548519.90
      2440240.77     13547827.18
#Sta/Elev= 30
  3973.2  307.48  4135.1  302.55  4338.4  297.73  4358.5  297.90  4379.2  296.29
  4429.1  295.84  4469.4  293.90  4519.8  293.69  4620.7  290.83  4791.9  287.68
  4926.9  286.66  4983.6  283.58  5006.6  283.33  5018.5  282.07  5019.0  281.57
  5029.4  282.07  5034.0  284.84  5039.1  286.80  5078.6  286.13  5085.4  286.81
  5118.6  287.23  5255.4  287.74  5283.8  288.85  5305.1  288.18  5425.0  287.71
  5587.7  288.42  5771.9  291.05  5849.6  292.65  5885.2  294.24  6056.3  295.88
#Mann=6,-1,0
  3973.2    0.05       0  4791.9    0.12       0  5018.5    0.05       0
  5029.4    0.12       0  5118.6    0.05       0  5305.1   0.035       0
Bank Sta=5018.5,5029.4
Exp/Cntr=0.3,0.1

Type RM Length L Ch R = 1,4685,435,435,435
BEGIN DESCRIPTION:
TRIB 3 TO YORKTOWN CREEK 6.0
END DESCRIPTION:
XS GIS Cut Line= 3
      2441675.00     13548925.02      2441525.00     13548275.00
      2440325.04     13547675.02
#Sta/Elev= 30
  4328.6  296.27  4352.6  294.42  4390.2  294.66  4480.8  291.54  4492.8  291.88
  4636.5  287.80  4842.9  285.58  4893.1  285.29  4913.6  283.53  4954.6  283.15
  4984.1  280.81  5004.2  280.29  5004.7  279.79  5015.2  280.29  5054.4  284.11
  5107.5  283.98  5115.9  282.67  5121.5  283.92  5129.9  284.38  5152.2  284.82
  5160.6  283.84  5183.0  286.68  5219.3  287.22  5384.2  284.71  5428.9  285.61
  5577.1  285.44  5842.5  287.62  6194.8  294.26  6233.9  295.84  6337.3  296.18
#Mann=6,-1,0
  4328.6    0.05       0  4842.9    0.12       0  4984.1    0.05       0
  5004.2    0.05       0  5015.2    0.05       0  5842.5   0.035       0
Bank Sta=5004.2,5015.2
Exp/Cntr=0.3,0.1

Type RM Length L Ch R = 1,4250,465,465,465
BEGIN DESCRIPTION:
Mapping XS 68f7227e
END DESCRIPTION:
XS GIS Cut Line= 3
      2441845.98     13548814.17      2441693.21     13547946.15
      2440978.98     13547394.87
#Sta/Elev= 30
  3968.8  294.12  3998.3  292.98  4003.4  293.52  4008.6  292.30  4039.0  291.48
  4294.9  286.92  4364.0  286.99  4467.7  284.82  4600.7  284.26  4841.2  284.07
  4907.0  285.04  4927.9  283.63  4942.4  281.31  4999.5  279.38  5005.9  278.30
  5015.7  275.81  5016.2  275.31  5026.7  275.81  5035.7  279.89  5042.0  280.58
  5056.5  284.19  5062.8  284.02  5071.0  285.16  5176.9  283.75  5220.4  280.46
  5234.9  282.84  5277.4  284.76  5560.1  287.46  5627.1  287.29  5752.4  288.83
#Mann=6,-1,0
  3968.8    0.05       0  4600.7    0.12       0  5005.9    0.05       0
  5015.7    0.05       0  5026.7    0.05       0  5560.1    0.12       0
Bank Sta=5015.7,5026.7
Exp/Cntr=0.3,0.1

Type RM Length L Ch R = 1,3785,502,502,502
BEGIN DESCRIPTION:
TRIB 3 TO YORKTOWN CREEK 5.0
END DESCRIPTION:
XS GIS Cut Line= 3
      2442025.00     13548774.97      2441925.00     13547575.00
      2441474.98     13547024.97
#Sta/Elev= 30
  3760.7  293.08  3810.8  290.90  4051.7  287.11  4300.0  284.28  4402.9  284.32
  4420.4  283.33  4556.1  282.61  4703.9  282.53  4872.5  283.91  4944.8  282.75
  4962.3  280.24  4968.1  280.24  4995.2  273.40  4995.7  272.90  5006.2  273.40
  5007.2  275.74  5029.4  278.10  5056.7  279.59  5093.3  279.95  5099.8  280.79
  5114.1  279.56  5147.2  278.69  5149.3  278.81  5157.2  275.99  5163.7  275.87
  5192.4  280.11  5213.2  281.96  5221.1  283.66  5578.5  290.06  5675.5  292.33
#Mann=7,-1,0
  3760.7    0.05       0  4556.1    0.12       0  4872.5    0.05       0
  4995.2    0.05       0  5006.2    0.05       0  5147.2    0.05       0
  5578.5   0.013       0
Bank Sta=4995.2,5006.2
Exp/Cntr=0.3,0.1

Type RM Length L Ch R = 1,3283,215,215,215
BEGIN DESCRIPTION:
Mapping XS 5f9ed00f
END DESCRIPTION:
XS GIS Cut Line= 4
      2442210.57     13548755.15      2442339.04     13547567.67
      2442231.40     13547338.51      2441672.39     13546935.74
#Sta/Elev= 30
  3756.5  291.58  4269.6  282.73  4319.9  283.35  4450.7  280.96  4712.2  280.49
  4775.7  280.82  4853.0  283.94  4928.5  283.25  4933.5  282.70  4943.5  278.83
  4949.7  273.73  4955.1  273.73  4964.9  270.42  4970.7  269.96  4971.2  269.46
  4983.0  269.96  4994.1  273.77  5009.1  275.66  5036.3  275.99  5053.3  277.04
  5075.4  280.54  5113.7  282.12  5159.3  282.83  5179.0  280.18  5219.8  280.21
  5268.7  281.97  5419.6  282.69  5668.3  286.91  5815.1  289.86  5893.1  291.99
#Mann=9,-1,0
  3756.5    0.05       0  4928.5     0.1       0  4970.7    0.05       0
  4983.0     0.1       0  5036.3    0.04       0  5179.0    0.05       0
  5219.8    0.04       0  5668.3    0.05       0  5815.1   0.013       0
Bank Sta=4970.7,4983
Exp/Cntr=0.3,0.1
