--- TRIB 4 TO EIGHTEENMILE CREEK.prj (project) ---

Proj Title=TRIB 4 TO EIGHTEENMILE CREEK Base Level Engineering
Current Plan=p01
Default Exp/Contr=0.3,0.1
English Units
Geom File=g01
Flow File=f01
Plan File=p01
Y Axis Title=Elevation
X Axis Title(PF)=Main Channel Distance
X Axis Title(XS)=Station
BEGIN DESCRIPTION:
TRIB 4 TO EIGHTEENMILE CREEK
END DESCRIPTION:
DSS Export Rating Curves= 0
DSS Export Rating Curve Sorted= 0
DSS Export Volume Flow Curves= 0
DXF OffsetX= 0
DXF OffsetY= 0
DXF ScaleX= 1
DXF ScaleY= 10

--- TRIB 4 TO EIGHTEENMILE CREEK.p01 (plan) ---

Plan Title=Multiple Run
Short Identifier=Multiple
Geom File=g01
Flow File=f01
Subcritical Flow
K Sum by GR= 0
Std Step Tol= 0.01
Critical Tol= 0.01
Num of Std Step Trials= 20
Max Error Tol= 0.3
Flow Tol Ratio= 0.001
Split Flow NTrial= 30
Split Flow Tol= 0.02
Split Flow Ratio= 0.02
Log Output Level= 0
Friction Slope Method= 1
Unsteady Friction Slope Method= 2
Unsteady Bridges Friction Slope Method= 1
Parabolic Critical Depth
Global Vel Dist=  1 , 1 , 1
Global Log Level= 0
CheckData=True
Encroach Param= -1, 0, 0, 0
BEGIN DESCRIPTION:
Multiple Run
END DESCRIPTION:

--- TRIB 4 TO EIGHTEENMILE CREEK.f01 (steady flow) ---

Flow Title=Multiple
Number of Profiles=7
Profile Names=10-year,25-year,50-year,1pct_min,100-year,1pct_plu,500-year
River Rch & RM= TRIB 4 TO EIGHTE,Reach-1,19144
     256     388     499     313     624    1245     960
River Rch & RM= TRIB 4 TO EIGHTE,Reach-1,16147
     730    1178    1582    1028    2050    4091    3408
River Rch & RM= TRIB 4 TO EIGHTE,Reach-1,9318
    2140    3632    5043    3375    6733   13435   11889
River Rch & RM= TRIB 4 TO EIGHTE,Reach-1,4713
    2393    4079    5681    3811    7604   15172   13497
Boundary for River Rch & Prof#=TRIB 4 TO EIGHTE,Reach-1,1
Up Type=0
Dn Type=3
Dn Slope=0.005
Boundary for River Rch & Prof#=TRIB 4 TO EIGHTE,Reach-1,2
Up Type=0
Dn Type=3
Dn Slope=0.005
Boundary for River Rch & Prof#=TRIB 4 TO EIGHTE,Reach-1,3
Up Type=0
Dn Type=3
Dn Slope=0.005
Boundary for River Rch & Prof#=TRIB 4 TO EIGHTE,Reach-1,4
Up Type=0
Dn Type=3
Dn Slope=0.005
Boundary for River Rch & Prof#=TRIB 4 TO EIGHTE,Reach-1,5
Up Type=0
Dn Type=3
Dn Slope=0.005
Boundary for River Rch & Prof#=TRIB 4 TO EIGHTE,Reach-1,6
Up Type=0
Dn Type=3
Dn Slope=0.005
Boundary for River Rch & Prof#=TRIB 4 TO EIGHTE,Reach-1,7
Up Type=0
Dn Type=3
Dn Slope=0.005

--- TRIB 4 TO EIGHTEENMILE CREEK.g01 (geometry) ---

Geom Title=Existing Conditions
Program Version=4.10

River Reach=TRIB 4 TO EIGHTE,Reach-1
Reach XY= 30
        2493875.       13484575.      2493425.37     13486359.73
      2494268.01     13488025.22      2494075.37     13488240.27
      2494175.32     13488600.11      2493973.04     13490419.35
      2493624.91     13490790.36      2493779.99     13491427.62
      2494025.26     13491494.94      2493778.36     13491676.25
      2493728.54     13492173.54      2494318.81     13492767.25
      2494564.65     13492764.76      2494533.25     13493271.93
      2495305.02     13493425.04      2495823.54     13493178.53
      2496024.26     13493435.69      2495875.37     13493690.17
      2495968.93     13493916.87      2496440.16     13494174.62
      2497073.55     13494028.53      2497268.81     13494417.19
      2497619.11     13494376.97      2498041.67     13494641.65
      2498171.57     13494923.78      2497826.56     13495118.92
      2498465.71     13495368.31      2498467.25     13495581.19
      2498074.52     13495940.16        2498475.       13496425.

Type RM Length L Ch R = 1 ,19144   ,231,231,231
BEGIN DESCRIPTION:
TRIB 4 TO EIGHTEENMILE CREEK 37.0
END DESCRIPTION:
XS GIS Cut Line= 3
      2493574.96     13484474.98      2493883.32     13484631.04
      2494340.34     13484545.27
#Sta/Elev= 30
  4654.4  250.53  4712.9  249.06  4721.7  249.24  4774.2  247.94  4824.3  246.47
  4855.8  244.74  4868.9  244.49  4891.2  243.23  4907.9  242.98  4913.5  242.07
  4930.1  240.75  5009.9  240.45  5010.1  239.95  5013.6  239.95  5013.9  240.45
  5022.1  241.19  5032.2  241.64  5042.4  242.86  5052.6  244.94  5058.8   246.7
  5067.6  246.31  5083.1  244.71  5093.3  244.66    5195  246.86  5268.7  248.13
  5306.9  248.56  5357.8  249.74  5384.2  249.76  5408.7   250.6    5465  251.38
#Mann= 6 ,-1 , 0
  4654.4     .05       0  4855.8      .1       0  5009.9     .05       0
  5013.9      .1       0  5067.6     .07       0  5268.7     .05       0
Bank Sta=5009.9,5013.9
XS Rating Curve= 0 ,0
Exp/Cntr=0.3,0.1

Type RM Length L Ch R = 1 ,18913   ,185,185,185
BEGIN DESCRIPTION:
Mapping XS c51b62ad
END DESCRIPTION:
XS GIS Cut Line= 4
      2493400.97     13484645.03      2493832.84     13484812.14
      2494019.47     13484825.16      2494347.17     13484653.71
#Sta/Elev= 30
    4532   246.3  4628.2  246.73  4633.5  246.36  4652.8  246.47  4736.7   245.3
  4763.5  244.49  4772.5  244.08  4782.9   244.3  4797.1  243.54  4846.2  242.94
  4904.7  240.48  4943.8  239.51  4960.6  240.39    4966  239.91  4975.9  240.29
  4991.5  239.27  4991.8  238.77  4995.3  238.77  4995.5  239.27  5017.3  239.43
  5067.4  240.94  5106.5  241.23  5110.3  240.99  5117.5  241.56  5208.2  243.16
  5262.9  244.11  5320.4  245.66  5433.4  247.71  5541.2  249.87    5552   249.8
#Mann= 10 ,-1 , 0
    4532     .05       0  4736.7    .035       0  4763.5     .05       0
  4904.7      .1       0  4991.5     .05       0  4995.5      .1       0
  5106.5     .07       0  5208.2    .035       0  5262.9     .07       0
  5433.4    .035       0
Bank Sta=4991.5,4995.5
XS Rating Curve= 0 ,0
Exp/Cntr=0.3,0.1

Type RM Length L Ch R = 1 ,18728   ,240,240,240
BEGIN DESCRIPTION:
Mapping XS b99a22ce
END DESCRIPTION:
XS GIS Cut Line= 3
      2493416.17     13484866.39      2493800.28     13484990.09
       2494211.3      13484983.6
#Sta/Elev= 30
  4586.6  241.69  4599.7  241.59  4626.6  242.06  4631.8  241.79  4658.6  241.87
  4663.9  241.55  4690.4  241.54  4733.3  240.61  4757.1  240.49  4816.5   239.7
  4827.8  239.22  4888.4  238.46  4942.2  237.02  4984.6  236.89    4988  236.03
  4988.2  235.53  4991.7  235.53    4992  236.03  5030.8  237.62  5054.9  238.55
  5114.9  239.22  5129.2  239.65  5154.9  240.78  5264.9  243.06  5284.9  243.79
  5293.8  243.73  5354.9  244.58  5364.9  245.05  5384.9  245.09  5401.2  245.61
#Mann= 9 ,-1 , 0
  4586.6     .05       0  4757.1    .035       0  4827.8      .1       0
  4942.2     .05       0    4988     .05       0    4992     .05       0
  5030.8    .035       0  5129.2     .05       0  5293.8     .07       0
Bank Sta=4988,4992
XS Rating Curve= 0 ,0
Exp/Cntr=0.3,0.1

Type RM Length L Ch R = 1 ,18488   ,83,83,83
BEGIN DESCRIPTION:
Mapping XS 8616b350
END DESCRIPTION:
XS GIS Cut Line= 3
       2493138.4     13485137.66      2493737.35     13485198.42
      2494321.12     13485220.12
#Sta/Elev= 30
  4410.2  245.96  4432.6  245.02  4437.7   245.1  4547.5  241.79  4650.2   238.4
    4716  236.81  4818.9  234.96    4835  234.95  4841.1   234.8  4899.3   235.7
  4919.4  235.28  4931.6  234.53  4989.8  234.69  5006.5  234.24  5006.8  233.74
  5010.3  233.74  5010.5  234.24  5049.8  234.59  5054.8  234.27  5060.4  234.38
  5061.1  234.39    5220  237.96  5270.1   238.6  5410.1   241.4  5450.2     242
  5460.2  241.76  5500.2  242.46  5520.2  242.35  5550.2   243.1  5596.4   243.4
#Mann= 9 ,-1 , 0
  4410.2     .05       0  4650.2     .07       0    4716     .05       0
    4835    .035       0  4841.1     .05       0  5006.5     .05       0
  5010.5     .05       0  5060.4    .035       0  5061.1     .05       0
Bank Sta=5006.5,5010.5
XS Rating Curve= 0 ,0
Exp/Cntr=0.3,0.1

Type RM Length L Ch R = 1 ,18405   ,404,404,404
BEGIN DESCRIPTION:
Mapping XS 888f33d0
END DESCRIPTION:
XS GIS Cut Line= 3
      2493144.86     13485311.27      2493711.31     13485278.72
      2494231.02     13485315.53
#Sta/Elev= 30
  4425.5  245.28  4449.2  245.07  4515.8  242.59  4585.9  240.78  4621.6  239.28
  4676.1  237.92  4706.1  236.71  4726.1  236.52  4793.7  234.36  4821.2  233.87
  4836.3  233.68  4884.4  232.08  4884.6  231.58  4888.1  231.58  4888.4  232.08
  4926.5  233.05    5016  233.07  5056.7  234.06  5066.8  233.84  5076.8  234.11
  5086.8  235.02  5096.8  235.24  5106.9  234.46  5152.3  236.03  5157.3  235.67
  5293.2  238.05  5298.2  237.78  5407.6  239.23  5439.2  238.77  5513.9  240.33
#Mann= 6 ,-1 , 0
  4425.5     .07       0  4621.6      .1       0  4821.2     .12       0
  4884.4     .05       0  4888.4     .12       0    5016     .05       0
Bank Sta=4884.4,4888.4
XS Rating Curve= 0 ,0
Exp/Cntr=0.3,0.1

Type RM Length L Ch R = 1 ,18001   ,310,310,310
BEGIN DESCRIPTION:
Mapping XS 9ffaa928
END DESCRIPTION:
XS GIS Cut Line= 3
      2493179.58     13485534.78      2493555.06     13485630.28
      2494230.01     13485612.92
#Sta/Elev= 30
  4600.5  241.53  4621.6  241.21  4626.8  240.49  4688.6  238.63  4709.3  238.47
  4758.7  236.64  4780.1   235.7  4791.8  234.73  4802.1   234.8  4826.2  233.55
  4853.7  233.38  4874.4  232.21  4993.8  228.28  4994.1  227.78  4997.6  227.78
  4997.8  228.28  5022.1  228.72  5057.9  229.45  5087.9  229.29  5157.6  230.93
  5177.9  231.05  5207.9  232.19    5248  232.96    5268  234.11    5288  232.96
  5385.4  234.98  5419.5  235.52  5618.1  239.39  5638.1  240.21  5663.1   240.3
#Mann= 8 ,-1 , 0
  4600.5     .12       0  4758.7      .1       0  4993.8     .05       0
  4997.8      .1       0  5022.1      .1       0  5157.6     .05       0
  5385.4    .035       0  5419.5     .05       0
Bank Sta=4993.8,4997.8
XS Rating Curve= 0 ,0
Exp/Cntr=0.3,0.1

Type RM Length L Ch R = 1 ,17691   ,192,192,192
BEGIN DESCRIPTION:
Mapping XS 73347ad8
END DESCRIPTION:
XS GIS Cut Line= 3
      2492986.45     13485784.35      2493489.95     13485927.59
      2494047.64     13485873.34
#Sta/Elev= 30
  4445.7  237.74  4496.2  237.19  4541.2   235.9  4575.1  235.88  4580.3  235.35
  4589.7  235.46  4656.4  233.81  4793.9  230.53  4832.9  230.03  4849.7  229.28
  4944.9  226.99  4969.2  225.73  4974.3  224.57  4982.3  224.04  4982.5  223.54
    4986  223.54  4986.3  224.04  5024.5  226.85    5098  229.28  5145.1  230.48
  5165.1  231.41  5185.2  231.22  5275.7  233.77  5296.1  233.76  5315.9  233.61
  5335.9  235.34  5359.2  234.68  5386.2  236.05  5497.8  238.29  5529.5  238.92
#Mann= 7 ,-1 , 0
  4445.7     .12       0  4656.4      .1       0  4982.3     .05       0
  4986.3      .1       0    5098     .12       0  5296.1    .035       0
  5497.8     .05       0
Bank Sta=4982.3,4986.3
XS Rating Curve= 0 ,0
Exp/Cntr=0.3,0.1

Type RM Length L Ch R = 1 ,17499   ,237,237,237
BEGIN DESCRIPTION:
Mapping XS 9c91d4ec
END DESCRIPTION:
XS GIS Cut Line= 3
      2493025.54     13485957.97      2493472.59      13486101.2
      2493940.66     13486001.52
#Sta/Elev= 30
  4528.1  232.64    4539  232.19  4630.2  231.79  4653.5  230.95    4706  231.06
  4737.5  229.59  4842.6  228.16  4962.1  225.27  4995.5  222.14  4995.8  221.64
  4999.3  221.64  4999.5  222.14  5020.4  224.51  5048.7  226.03  5098.2  227.87
  5141.8  228.74  5214.7  230.95    5243  231.24  5255.6  231.66  5265.8  231.01
  5291.4   231.4  5296.5  232.22  5327.2  233.11  5344.1  233.03  5378.3  233.28
  5385.4  234.56  5398.7  234.98  5419.2  234.38  5429.4  235.12  5476.1  236.53
#Mann= 6 ,-1 , 0
  4528.1      .1       0  4995.5     .05       0  4999.5      .1       0
  5141.8     .07       0    5243     .12       0  5344.1    .035       0
Bank Sta=4995.5,4999.5
XS Rating Curve= 0 ,0
Exp/Cntr=0.3,0.1

Type RM Length L Ch R = 1 ,17262   ,373,373,373
BEGIN DESCRIPTION:
Mapping XS 50c15284
END DESCRIPTION:
XS GIS Cut Line= 3
      2492863.67     13486287.65       2493426.2     13486322.38
      2493835.96     13486162.64
#Sta/Elev= 30
  4438.4  235.39  4469.8  235.16  4499.8  233.36  4549.9  232.11    4560  232.23
    4600  230.29  4680.2  228.87  4710.2   227.8  4730.3  227.81  4798.3  226.26
  4820.5   226.3  4890.6   224.7  4959.6  221.67  4964.6  221.98  4970.7  220.78
  4980.8  219.68  4996.9  219.22  4997.1  218.72  5000.6  218.72  5000.9  219.22
    5004  219.22  5007.3  220.17  5022.2   222.1    5108  224.48  5197.8  226.09
  5333.4  228.66  5344.2   229.3  5411.2  230.81  5423.1  230.89  5441.8  232.13
#Mann= 5 ,-1 , 0
  4438.4      .1       0  4996.9     .05       0  5000.9      .1       0
  5197.8     .07       0  5411.2     .05       0
Bank Sta=4996.9,5000.9
XS Rating Curve= 0 ,0
Exp/Cntr=0.3,0.1

Type RM Length L Ch R = 1 ,16889   ,218,218,218
BEGIN DESCRIPTION:
Mapping XS 7d8ace20
END DESCRIPTION:
XS GIS Cut Line= 4
      2493051.18     13486627.93      2493578.98     13486641.82
      2493759.54     13486593.21      2494335.92     13486350.16
#Sta/Elev= 30
  4475.9  232.54  4589.8  229.95  4629.8  228.49  4764.3  224.88  4789.3  224.28
  4829.8  223.47  4924.2  220.57  4969.9  219.62  4989.9  217.69  5005.9  216.85
  5006.2  216.35  5009.7  216.35  5009.9  216.85  5013.1  217.31  5023.3  217.12
  5030.8  217.56  5047.9  219.93  5072.3  220.76    5093     222  5125.9  222.37
  5195.3  223.38  5353.9  226.87  5401.3  227.17  5413.9  227.81  5544.1  229.32
  5612.8  229.32  5636.5  228.69  5736.8  228.12  5765.9  228.47  5816.4  228.21
#Mann= 8 ,-1 , 0
  4475.9     .05       0  4764.3     .07       0  4789.3     .05       0
  4924.2     .07       0  5005.9     .05       0  5009.9     .07       0
  5023.3     .07       0  5125.9     .05       0
Bank Sta=5005.9,5009.9
XS Rating Curve= 0 ,0
Exp/Cntr=0.3,0.1

Type RM Length L Ch R = 1 ,16671   ,524,524,524
BEGIN DESCRIPTION:
Mapping XS 2afcf76b
END DESCRIPTION:
XS GIS Cut Line= 3
      2492838.95     13487008.31       2493646.2     13486839.05
      2494379.74      13486426.7
#Sta/Elev= 30
  4180.4   237.9  4266.3  235.43  4271.5  235.84  4425.4  232.34  4452.2  232.31
  4623.9  227.75    4753  224.17  4954.9  219.05    4976  217.91  4993.8  216.94
  4999.7  215.42  5000.9  214.26  5001.1  213.76  5004.9  214.26  5005.2  214.26
  5022.4  218.09  5056.6  218.34  5095.6  218.62  5175.9  220.88    5206  220.88
  5249.3  222.35  5302.1  222.39  5373.6  224.21    5417  223.98  5432.9  225.12
  5513.9  226.46  5573.2  226.17  5578.9  226.77  5756.8  225.03  5846.7  225.56
#Mann= 10 ,-1 , 0
  4180.4     .05       0  4266.3    .035       0  4425.4     .05       0
  4623.9    .035       0    4753     .05       0    4976     .07       0
  5000.9     .05       0  5004.9     .07       0  5005.2     .07       0
  5056.6     .05       0
Bank Sta=5000.9,5004.9
XS Rating Curve= 0 ,0
Exp/Cntr=0.3,0.1

Type RM Length L Ch R = 1 ,16147   ,237,237,237
BEGIN DESCRIPTION:
TRIB 4 TO EIGHTEENMILE CREEK 31.0
END DESCRIPTION:
XS GIS Cut Line= 3
        2493625.       13487275.        2493925.       13487225.
        2494525.       13487075.
#Sta/Elev= 30
  4700.3  220.97    4751  220.06  4904.4   215.8    5007  212.85  5014.7  212.53
  5025.6  210.99  5025.9  210.49  5029.4  210.49  5029.6  210.99  5055.6  213.09
  5076.6   213.8  5117.8  212.22  5157.7  213.64  5179.7  213.75  5187.4  213.22
  5192.6  213.73  5210.6  212.92  5223.4  214.22  5228.6  214.98  5233.8  214.84
  5241.5  215.66  5262.1  218.51  5269.9  220.08    5275     223  5311.1  223.03
  5316.2  222.35    5324  222.98  5352.3   219.4  5365.2  219.39  5622.9   225.8
#Mann= 7 ,-1 , 0
  4700.3     .05       0  4904.4      .1       0  5025.6     .05       0
  5029.6      .1       0  5055.6     .12       0  5157.7     .05       0
  5223.4     .07       0
Bank Sta=5025.6,5029.6
XS Rating Curve= 0 ,0
Exp/Cntr=0.3,0.1

Type RM Length L Ch R = 1 ,15910   ,248,248,248
BEGIN DESCRIPTION:
Mapping XS 0b8a91b4
END DESCRIPTION:
XS GIS Cut Line= 3
      2493498.61     13487424.98      2493971.72     13487446.69
      2494674.87     13487220.98
#Sta/Elev= 30
  4522.9  223.84  4526.7  223.62  4564.2  222.77  4599.4  221.63  4633.4  221.21
  4759.5  218.32  4894.7  213.94  4929.7  212.02  4949.7  212.12  4989.8  210.72
  4992.8  209.16  4993.7  208.69  4993.9  208.19  4997.4  208.19  4997.7  208.69
  5010.5  209.14  5017.1  210.26    5042  212.15    5063  212.17  5096.8  213.92
    5168  214.19  5199.5  215.13  5241.5  215.45  5367.5  218.18  5438.6  220.59
  5493.6  222.09  5556.6  224.55    5643  226.56  5682.6  228.09    5735  229.11
#Mann= 9 ,-1 , 0
  4522.9     .05       0  4526.7    .035       0  4564.2     .05       0
  4894.7      .1       0  4992.8     .12       0  4993.7     .05       0
  4997.7     .12       0  5096.8     .05       0  5438.6     .07       0
Bank Sta=4993.7,4997.7
XS Rating Curve= 0 ,0
Exp/Cntr=0.3,0.1

Type RM Length L Ch R = 1 ,15662   ,437,437,437
BEGIN DESCRIPTION:
TRIB 4 TO EIGHTEENMILE CREEK 30.0
END DESCRIPTION:
XS GIS Cut Line= 3
      2493724.99       13487625.        2494025.       13487675.
      2494625.02     13487374.99
#Sta/Elev= 30
  4695.9  218.93  4723.8  217.88    4777  216.53  4850.5   214.2  4868.3  214.05
  4890.4  213.26  4939.2     212  4959.5  210.75  4967.1  210.01  4972.2  210.45
  4979.8  209.49  4997.5  208.41  5002.8  208.41    5012  207.57  5012.3  207.07
  5015.8  207.07    5016  207.57  5022.4  208.73  5044.8  211.06  5062.6  211.24
  5075.5  211.19  5120.2  211.96  5151.1  212.12  5201.3  212.76  5335.5   215.8
  5438.9  218.97    5506  221.25  5514.3  221.74  5620.9  224.98  5670.9  226.63
#Mann= 7 ,-1 , 0
  4695.9     .05       0  4890.4      .1       0    5012     .05       0
    5016      .1       0  5062.6     .12       0  5151.1     .05       0
  5620.9     .07       0
Bank Sta=5012,5016
XS Rating Curve= 0 ,0
Exp/Cntr=0.3,0.1

Type RM Length L Ch R = 1 ,15225   ,459,459,459
BEGIN DESCRIPTION:
TRIB 4 TO EIGHTEENMILE CREEK 29.0
END DESCRIPTION:
XS GIS Cut Line= 3
      2493675.03     13487825.01        2494275.       13488025.
      2494575.01     13487724.99
#Sta/Elev= 30
  4375.4  219.93  4470.2  216.33  4480.8  216.22  4491.3   215.7  4533.5  214.56
  4596.7  212.13  4635.1   211.7  4754.8  208.88  4814.2  208.57  4860.2  208.48
  4891.9  207.83    4913  207.85    4934  206.77  4955.1  206.48  4963.7  206.09
  4963.9  205.59  4967.4  205.59  4967.7  206.09  5005.2  207.45    5022   207.1
  5064.4  207.73  5078.5  208.18  5092.7  209.13  5106.8  210.77  5149.2  211.39
  5163.4  212.18  5190.6  212.96  5333.1  216.33  5361.4  217.57  5432.1  219.43
#Mann= 6 ,-1 , 0
  4375.4     .05       0  4635.1     .07       0  4814.2      .1       0
  4963.7     .05       0  4967.7      .1       0  5190.6     .05       0
Bank Sta=4963.7,4967.7
XS Rating Curve= 0 ,0
Exp/Cntr=0.3,0.1

Type RM Length L Ch R = 1 ,14766   ,459,459,459
BEGIN DESCRIPTION:
TRIB 4 TO EIGHTEENMILE CREEK 28.0
END DESCRIPTION:
XS GIS Cut Line= 3
      2493524.98     13487974.99        2494125.       13488375.
      2494724.97       13488375.
#Sta/Elev= 30
  4288.7   222.1  4396.9   219.2  4561.8  213.33  4569.8  213.14  4605.7   211.7
  4677.7  210.15  4698.9  209.47  4728.9  209.87  4743.9  208.83  4793.5  207.98
  4799.7  207.34  4901.7  206.18  4937.7  206.83  4945.2  204.98  4960.3  204.62
  4981.3  205.12  5037.8  204.51  5038.1  204.01  5041.6  204.01  5041.8  204.51
  5049.8     205  5069.8  208.12  5089.8  206.68  5155.3   207.3  5229.8  210.46
  5339.8   212.7  5416.4  215.18  5509.8  218.63  5539.8  218.91  5609.8  221.78
#Mann= 9 ,-1 , 0
  4288.7     .05       0  4561.8     .07       0  4569.8    .035       0
  4677.7     .07       0  4799.7      .1       0  5037.8     .05       0
  5041.8      .1       0  5155.3     .07       0  5416.4     .12       0
Bank Sta=5037.8,5041.8
XS Rating Curve= 0 ,0
Exp/Cntr=0.3,0.1

Type RM Length L Ch R = 1 ,14307   ,451,451,451
BEGIN DESCRIPTION:
TRIB 4 TO EIGHTEENMILE CREEK 27.0
END DESCRIPTION:
XS GIS Cut Line= 3
      2493524.98     13488324.98        2494075.       13488775.
      2494675.02     13489075.01
#Sta/Elev= 30
    4290  218.05  4445.7  214.61  4569.8  210.87  4610.2  209.42  4659.7  208.88
  4716.4  206.97    4781  206.29  4801.8  205.36  4936.1  204.31  4979.1  202.83
  4991.5  201.67  4991.7  201.17  4995.2  201.17  4995.5  201.67  4997.4  203.25
    5009  203.87  5059.4  203.39  5143.2   203.9  5148.8  203.43  5165.6  205.09
  5193.5  204.96  5215.9  206.33  5247.8   207.2  5327.7   210.6  5372.4   211.8
  5425.5  214.67  5439.5  214.75  5470.2  216.59    5600  221.84  5671.5  224.22
#Mann= 7 ,-1 , 0
    4290     .07       0  4445.7    .035       0  4569.8      .1       0
  4991.5     .05       0  4995.5      .1       0  5247.8     .12       0
    5600     .05       0
Bank Sta=4991.5,4995.5
XS Rating Curve= 0 ,0
Exp/Cntr=0.3,0.1

Type RM Length L Ch R = 1 ,13856   ,443,443,443
BEGIN DESCRIPTION:
TRIB 4 TO EIGHTEENMILE CREEK 26.0
END DESCRIPTION:
XS GIS Cut Line= 3
      2493424.97       13489075.        2493975.       13489125.
        2494575.       13489125.
#Sta/Elev= 30
  4443.5  211.91  4664.4  205.71  4744.8  204.45  4764.9  204.57  4774.9  203.71
    4795  204.55  4821.1  204.02  4915.5  203.37  4935.6  202.68  4955.6  203.16
  4985.8  202.37  5013.8  200.43  5014.1  199.93  5017.6  199.93  5017.8  200.43
  5035.8  202.01  5055.8  201.83  5085.8  202.58  5105.8  202.57  5135.8  201.39
  5220.8  205.24  5245.8  206.46  5255.8  206.34  5275.8  207.51  5325.8  208.76
  5385.8  211.81  5445.8  213.42  5495.8  216.34  5525.8  217.13  5595.8  220.85
#Mann= 5 ,-1 , 0
  4443.5     .12       0  4821.1      .1       0  5013.8     .05       0
  5017.8      .1       0  5220.8     .12       0
Bank Sta=5013.8,5017.8
XS Rating Curve= 0 ,0
Exp/Cntr=0.3,0.1

Type RM Length L Ch R = 1 ,13413   ,452,452,452
BEGIN DESCRIPTION:
TRIB 4 TO EIGHTEENMILE CREEK 25.0
END DESCRIPTION:
XS GIS Cut Line= 3
      2493425.01     13489125.01        2494025.       13489525.
      2494324.97     13489475.01
#Sta/Elev= 30
  4278.5  211.74  4358.1  209.22  4364.1  209.51  4386.6  208.98  4400.2  208.12
  4487.3  205.65  4494.8   206.1  4502.3  205.45  4517.4  205.31    4566  203.14
  4631.5   201.8  4652.6  202.35  4675.1  201.48  4821.3  200.95    4854  200.54
  4862.9  201.04  4883.9  200.47  4927.5  200.62    4956  200.06  4992.1  200.72
  5002.1   200.5  5007.7  199.37    5008  198.87  5011.5  198.87  5011.7  199.37
  5019.9  200.22  5102.1  202.87  5263.2  208.24  5283.5   209.6  5303.7  210.24
#Mann= 7 ,-1 , 0
  4278.5     .12       0    4566      .1       0  4821.3     .12       0
    4854      .1       0  5007.7     .05       0  5011.7      .1       0
  5102.1     .12       0
Bank Sta=5007.7,5011.7
XS Rating Curve= 0 ,0
Exp/Cntr=0.3,0.1

Type RM Length L Ch R = 1 ,12961   ,484,484,484
BEGIN DESCRIPTION:
TRIB 4 TO EIGHTEENMILE CREEK 24.0
END DESCRIPTION:
XS GIS Cut Line= 3
      2493375.03     13489325.03        2493975.       13489925.
      2494574.99     13490274.99
#Sta/Elev= 30
  4151.5  209.79  4278.7  205.67  4519.2  200.34    4604  199.85  4632.3  199.19
  4733.8  199.49  4787.9  198.91  4816.1  199.74  4886.9  199.69  4943.4   198.7
  4985.8  199.44  5002.9  198.65  5011.6  196.68  5011.9  196.18  5015.4  196.18
  5015.6  196.68  5029.3  198.62  5057.9  199.41  5115.8  199.94    5220  202.06
  5232.8  201.73  5303.3  203.48  5381.6   205.8  5446.1  209.39  5451.9  208.86
  5461.8  209.02  5474.7  210.36  5532.5  213.02  5547.8  213.22  5694.6  219.05
#Mann= 5 ,-1 , 0
  4151.5     .12       0  4733.8      .1       0  5011.6     .05       0
  5015.6      .1       0  5303.3     .07       0
Bank Sta=5011.6,5015.6
XS Rating Curve= 0 ,0
Exp/Cntr=0.3,0.1

Type RM Length L Ch R = 1 ,12477   ,446,446,446
BEGIN DESCRIPTION:
TRIB 4 TO EIGHTEENMILE CREEK 23.0
END DESCRIPTION:
XS GIS Cut Line= 3
        2493075.       13489975.        2493975.       13490375.
      2494174.97     13490424.99
#Sta/Elev= 30
  4014.6  209.63  4091.2  207.95    4122  206.62  4202.7  205.37  4211.6   204.3
  4233.5  203.32  4243.8  203.56  4371.2  200.38  4394.2  199.26  4440.7   199.2
  4452.3  198.32  4526.3  196.63  4573.4  195.57  4596.6  196.22  4627.4  195.35
  4649.3  196.38  4702.4  196.49    4819  196.13  4933.1  196.39  4967.3  195.45
  4977.6  195.94  4990.6  195.12  5002.1  196.04  5007.8  194.85    5008  194.35
  5011.8  194.85  5058.8  199.63  5105.1  201.19    5203  206.03  5205.6  206.04
#Mann= 9 ,-1 , 0
  4014.6     .12       0  4243.8     .07       0  4371.2     .12       0
  4526.3      .1       0  4702.4     .07       0    4819     .05       0
  5007.8     .05       0  5011.8     .05       0    5203     .07       0
Bank Sta=5007.8,5011.8
XS Rating Curve= 0 ,0
Exp/Cntr=0.3,0.1

Type RM Length L Ch R = 1 ,12031   ,442,442,442
BEGIN DESCRIPTION:
TRIB 4 TO EIGHTEENMILE CREEK 22.0
END DESCRIPTION:
XS GIS Cut Line= 3
      2492924.99       13490225.        2493675.       13490625.
      2494474.96       13490525.
#Sta/Elev= 30
    4142     211  4441.1  202.04  4464.7  201.28  4517.8  200.16  4534.1  198.92
    4670  195.85  4769.9  194.43  4779.7     195    4822  194.11  4867.3  195.31
  4920.1  194.58  4941.4  193.82  4983.9  194.49  4994.5  193.83  5002.1  191.46
  5010.2  190.72  5010.4  190.22  5014.2  190.72  5029.8  192.62  5034.8  192.26
  5052.5  193.97    5098   194.2  5197.4  194.65  5197.7  194.65    5254  194.54
  5271.7  196.25  5315.7  198.63    5506  207.82  5717.6  215.68  5798.2     218
#Mann= 13 ,-1 , 0
    4142     .12       0  4441.1     .07       0  4464.7     .05       0
    4670     .12       0  4779.7      .1       0  4920.1     .12       0
  4941.4      .1       0  5010.2     .05       0  5014.2      .1       0
    5098     .05       0  5197.4      .1       0  5197.7     .05       0
  5315.7     .07       0
Bank Sta=5010.2,5014.2
XS Rating Curve= 0 ,0
Exp/Cntr=0.3,0.1

Type RM Length L Ch R = 1 ,11589   ,461,461,461
BEGIN DESCRIPTION:
TRIB 4 TO EIGHTEENMILE CREEK 21.0
END DESCRIPTION:
XS GIS Cut Line= 3
      2492924.99     13490374.99        2493675.       13490975.
      2494474.99       13490575.
#Sta/Elev= 30
  4029.7  208.96  4044.5  208.97  4091.1  207.71  4136.2  206.34  4150.6  206.62
  4193.7  204.83  4256.9  202.84  4421.1  197.54  4460.1  196.92  4563.6  194.79
  4679.9  193.54  4826.1  192.02  4875.7  193.26  4890.1  192.61  4926.1  193.11
  4954.2  192.84  4985.9  191.28  5024.5   191.2  5024.7   190.7  5028.6   191.2
  5155.1  193.34  5177.5  194.71  5205.4   194.9  5339.6  198.85  5473.7  204.17
  5624.7  208.46  5781.2  214.16  5809.1  214.56  5831.5  216.06  5884.6  217.33
#Mann= 10 ,-1 , 0
  4029.7     .12       0  4044.5     .07       0  4091.1     .12       0
  4193.7     .05       0  4256.9     .07       0  4460.1     .05       0
  4679.9      .1       0  4985.9     .07       0  5024.5     .05       0
  5028.6     .07       0
Bank Sta=5024.5,5028.6
XS Rating Curve= 0 ,0
Exp/Cntr=0.3,0.1

Type RM Length L Ch R = 1 ,11128   ,456,456,456
BEGIN DESCRIPTION:
TRIB 4 TO EIGHTEENMILE CREEK 20.0
END DESCRIPTION:
XS GIS Cut Line= 3
      2492975.03     13491175.01        2493775.       13491375.
      2494575.01     13490874.99
#Sta/Elev= 30
  4167.5  205.09  4170.3  205.09  4270.9  203.04  4507.6  198.09  4765.8  189.14
  4766.1  188.64  4769.9  189.14  4812.8  190.92  4919.9  191.89  4940.5  191.34
  4961.2  189.68    4974  189.63  4981.8  189.79  5063.4  190.35    5100  189.88
    5328  196.45  5377.1  198.48  5507.3  201.96  5535.1   202.2  5617.1  206.61
  5623.6  206.84  5629.5  205.87  5660.1  208.04  5680.4  208.41  5685.2  208.58
  5696.7  209.12  5702.6  207.91  5739.1  209.74  5863.2  213.83  5935.5  215.95
#Mann= 14 ,-1 , 0
  4167.5     .05       0  4170.3    .035       0  4270.9     .05       0
  4765.8     .07       0  4769.9     .05       0  4812.8      .1       0
  4961.2     .05       0    4974     .07       0  4981.8      .1       0
    5328     .05       0  5507.3    .035       0  5680.4     .05       0
  5685.2    .035       0  5863.2     .07       0
Bank Sta=4961.2,4974
XS Rating Curve= 0 ,0
Exp/Cntr=0.3,0.1

Type RM Length L Ch R = 1 ,10672   ,901,901,901
BEGIN DESCRIPTION:
TRIB 4 TO EIGHTEENMILE CREEK 19.0
END DESCRIPTION:
XS GIS Cut Line= 3
      2493025.02       13491375.        2494025.       13491575.
        2494325.       13491325.
#Sta/Elev= 30
  3983.9  202.79  4086.2  202.07  4320.4  197.09  4463.2  192.62    4504  193.82
  4514.2  193.08  4529.1  190.29  4544.8  187.33  4575.4  187.06  4595.8   187.5
  4616.2  189.18  4677.3  190.65  4697.7  190.18  4758.9  191.64  4827.4  190.63
  4860.9  188.75  5015.3  186.95  5015.6  186.45  5019.4  186.95  5031.7  187.37
  5039.5  189.16    5046  188.55  5053.8  190.04  5068.1  191.29  5088.9  192.27
  5185.3  194.71    5210   196.2    5238  196.22  5344.1  201.18  5394.2   202.7
#Mann= 7 ,-1 , 0
  3983.9     .07       0  4086.2     .05       0  4529.1      .1       0
  4827.4    .035       0  5015.3    .035       0  5019.4    .035       0
  5185.3     .05       0
Bank Sta=5015.3,5019.4
XS Rating Curve= 0 ,0
Exp/Cntr=0.3,0.1

Type RM Length L Ch R = 1 ,9771    ,453,453,453
BEGIN DESCRIPTION:
TRIB 4 TO EIGHTEENMILE CREEK 18.0
END DESCRIPTION:
XS GIS Cut Line= 3
      2493174.97     13491824.98        2493775.       13492225.
      2494574.99     13491425.01
#Sta/Elev= 30
  4280.3  196.98  4424.6  195.18  4604.8  192.08  4792.6  186.88  4849.7  185.97
  4929.3  185.47  4936.9  184.39  4942.9  184.96  4951.9   183.7  4957.9  184.34
  4972.9  182.78  4981.6  182.73  4991.8   182.2  4992.1   181.7  4995.8   181.7
    4996   182.2  4998.4  182.69  5015.6  183.24  5043.9   183.1  5128.7  185.65
  5260.3  186.85  5397.4  187.89  5455.5  187.85  5581.3  189.05  5609.6  189.76
  5623.7  190.89    5652  190.91  5793.4  194.37  5835.8  196.62  6132.8  205.12
#Mann= 6 ,-1 , 0
  4280.3     .05       0  4981.6      .1       0  4991.8     .05       0
    4996      .1       0  5260.3     .12       0  5455.5     .05       0
Bank Sta=4991.8,4996
XS Rating Curve= 0 ,0
Exp/Cntr=0.3,0.1

Type RM Length L Ch R = 1 ,9318    ,439,439,439
BEGIN DESCRIPTION:
TRIB 4 TO EIGHTEENMILE CREEK 17.0
END DESCRIPTION:
XS GIS Cut Line= 3
      2493024.98     13493175.01        2494125.       13492475.
        2494875.       13492025.
#Sta/Elev= 30
  3690.1  197.59  3828.1  194.49  3943.3  190.24  4067.7  190.17  4306.5  184.47
    4480  184.41  4531.7  186.18  4570.9  184.68  4602.8  183.83  4689.2  184.59
  4834.8  182.95  4922.8  182.94  4986.3   181.9  4996.9  181.41  5001.4  180.49
  5001.9  179.99  5013.8  180.49  5038.7  181.52    5060  184.88  5144.4  186.06
  5271.9  186.42  5299.1  187.37  5308.8  186.71  5388.5  187.19  5505.1     190
  5600.4  194.27  5658.7   198.8  5680.1  198.25  5759.8  201.34  5868.6  204.28
#Mann= 5 ,-1 , 0
  3690.1     .05       0  4570.9      .1       0  5001.4     .05       0
  5013.8      .1       0  5144.4     .05       0
Bank Sta=5001.4,5013.8
XS Rating Curve= 0 ,0
Exp/Cntr=0.3,0.1

Type RM Length L Ch R = 1 ,8879    ,453,453,453
BEGIN DESCRIPTION:
TRIB 4 TO EIGHTEENMILE CREEK 16.0
END DESCRIPTION:
XS GIS Cut Line= 3
      2493975.02     13493424.96        2494375.       13492775.
        2494875.       13492175.
#Sta/Elev= 30
  4237.8   194.1  4262.8  193.75  4318.8  193.27  4398.1  190.35  4419.4  190.55
  4593.7  187.04  4709.3  184.71  4813.1  180.26  4834.8  181.27    4856  180.87
  4942.3  182.49  4956.6  182.06  4965.7  179.49    4987  178.31  4987.5  177.81
  4999.5  178.31    5001   179.9  5008.1   180.8  5052.9   181.9  5116.4  182.42
  5178.7  184.21  5211.8  183.77  5237.7  184.03  5384.3  185.22  5441.6  186.68
    5590  193.35  5647.3  196.55  5668.1   198.8  5682.4  197.89    5782  201.85
#Mann= 9 ,-1 , 0
  4237.8     .05       0  4262.8     .12       0  4593.7      .1       0
    4987     .05       0  4999.5      .1       0  5052.9    .035       0
  5116.4      .1       0  5211.8    .035       0  5237.7     .05       0
Bank Sta=4987,4999.5
XS Rating Curve= 0 ,0
Exp/Cntr=0.3,0.1

Type RM Length L Ch R = 1 ,8426    ,459,459,459
BEGIN DESCRIPTION:
TRIB 4 TO EIGHTEENMILE CREEK 15.0
END DESCRIPTION:
XS GIS Cut Line= 3
      2494074.98     13493475.02        2494625.       13492975.
      2494974.98     13492175.04
#Sta/Elev= 30
  4261.1  193.96  4395.9  192.16  4593.9  185.38  4622.5  185.24  4679.1  182.93
  4693.3  177.37  4693.8  175.51  4694.3  175.01  4706.3  175.51  4756.8  181.27
  4785.2  180.09  4791.9  178.01  4813.5  176.72  4827.7  177.43  4834.5  179.36
    4948  181.06    4969  180.79  4990.6  178.01  4997.3  178.08  5001.9  178.52
  5065.6  181.82    5188  182.76  5222.7  182.04  5334.9  183.68  5467.2  186.56
    5613  191.68  5665.2  193.83    5712  198.51  5724.8  197.98  5877.6  203.46
#Mann= 8 ,-1 , 0
  4261.1     .12       0  4622.5      .1       0  4693.8     .07       0
  4706.3      .1       0  4990.6     .05       0  4997.3     .07       0
  5001.9    .035       0  5334.9     .05       0
Bank Sta=4990.6,4997.3
XS Rating Curve= 0 ,0
Exp/Cntr=0.3,0.1

Type RM Length L Ch R = 1 ,7967    ,465,465,465
BEGIN DESCRIPTION:
TRIB 4 TO EIGHTEENMILE CREEK 14.0
END DESCRIPTION:
XS GIS Cut Line= 3
      2494074.96     13493575.02        2494575.       13493275.
      2495375.02     13492074.96
#Sta/Elev= 30
    4418   195.2  4431.6  195.81    4558  193.78  4906.1   183.2  4950.6  182.69
  4966.2  180.65  4977.8  175.49  4991.8  175.08  4992.3  174.58  5004.7  175.08
  5014.7  175.64  5023.7  177.49  5029.7  177.51  5037.2  179.55  5050.7  180.47
  5080.8  179.94  5145.4  181.12  5305.5   181.2  5433.8  181.97  5498.4  181.38
  5621.6  183.34  5735.8  185.78  6024.2   199.1  6183.5  202.75    6227  205.24
  6255.6  204.51  6327.7  205.56  6384.8  207.84  6407.3  209.61  6443.4   208.8
#Mann= 6 ,-1 , 0
    4418     .12       0  4906.1      .1       0  4991.8     .05       0
  5004.7      .1       0  5305.5    .035       0  5621.6     .05       0
Bank Sta=4991.8,5004.7
XS Rating Curve= 0 ,0
Exp/Cntr=0.3,0.1

Type RM Length L Ch R = 1 ,7502    ,468,468,468
BEGIN DESCRIPTION:
TRIB 4 TO EIGHTEENMILE CREEK 13.0
END DESCRIPTION:
XS GIS Cut Line= 3
        2494725.     13494124.99        2495025.       13493325.
      2495424.99     13492525.02
#Sta/Elev= 30
  4149.9  195.56  4206.7  195.17  4335.9  193.74  4391.1  191.97  4476.5  190.34
  4501.4  189.57    4537   187.4  4652.7  183.95  4738.2  183.08  4818.3  181.07
  4878.8  180.52  4909.1  178.85  4932.5   178.5  4964.2   177.5  4972.3  178.05
  4982.7  175.94  4983.2  175.44  4995.1  175.44  4995.6  175.94  5001.6  177.92
  5038.1  178.95  5101.8  179.48  5398.4  181.58  5532.6  183.95  5581.6  185.91
    5608  187.21  5638.8  189.69  5719.8  193.88  5810.4  196.94  5898.7  199.85
#Mann= 9 ,-1 , 0
  4149.9     .12       0  4206.7     .05       0  4932.5    .035       0
  4982.7    .035       0  4995.6    .035       0  5038.1      .1       0
  5101.8    .035       0  5581.6     .12       0  5810.4     .05       0
Bank Sta=4982.7,4995.6
XS Rating Curve= 0 ,0
Exp/Cntr=0.3,0.1

Type RM Length L Ch R = 1 ,7034    ,463,463,463
BEGIN DESCRIPTION:
TRIB 4 TO EIGHTEENMILE CREEK 12.0
END DESCRIPTION:
XS GIS Cut Line= 3
      2494824.99     13494125.01        2495425.       13493325.
        2495525.     13492724.99
#Sta/Elev= 30
  4010.4  196.34  4024.5  196.35  4096.9  195.87  4160.4   192.8  4332.3   187.9
    4474  184.76  4603.1   183.3  4746.9  179.27  4792.7  178.86    4874   179.9
  4888.5  179.52  4896.9  178.25  4903.1  178.79  4913.4  176.34  4917.7  175.36
    4924  175.84  4925.8  174.65  4926.3  174.15  4938.8  174.65    4974  175.47
  4982.3  176.47  5007.3  175.64  5012.9  175.64  5020.5  176.13  5121.9  177.04
  5172.6  179.77  5253.7  180.27  5328.4  182.26  5361.4  183.43  5618.7   195.6
#Mann= 11 ,-1 , 0
  4010.4    .035       0  4024.5     .05       0  4792.7    .035       0
  4913.4      .1       0  4925.8     .07       0  4938.8      .1       0
  5007.3     .05       0  5012.9     .07       0  5020.5      .1       0
  5328.4     .12       0  5361.4     .07       0
Bank Sta=5007.3,5012.9
XS Rating Curve= 0 ,0
Exp/Cntr=0.3,0.1

Type RM Length L Ch R = 1 ,6571    ,436,436,436
BEGIN DESCRIPTION:
TRIB 4 TO EIGHTEENMILE CREEK 11.0
END DESCRIPTION:
XS GIS Cut Line= 3
        2494925.       13494175.        2495825.       13493175.
      2495624.99     13492774.97
#Sta/Elev= 30
  3658.8  196.46  3736.9  195.22  3885.6  190.94  4281.8  183.04  4444.7  178.76
  4529.9  178.14  4559.2  178.76    4619  178.47  4706.9  177.97  4777.3  178.39
  4883.4   177.2  4947.7  175.09  4968.7  173.02  4969.6  172.38  4970.1  171.88
  4982.6  172.38  4997.1  175.32  5000.8  177.17    5007  177.17  5012.5  178.74
  5018.1  178.34  5034.9  179.84  5040.5  178.82  5048.9  179.84    5116  180.91
  5178.6  183.09  5290.4  188.21  5324.2  189.66  5353.5  191.29  5451.4  194.02
#Mann= 9 ,-1 , 0
  3658.8     .05       0  4559.2      .1       0    4619     .05       0
  4706.9      .1       0  4969.6     .05       0  4982.6      .1       0
  5178.6     .05       0  5290.4    .035       0  5324.2     .05       0
Bank Sta=4969.6,4982.6
XS Rating Curve= 0 ,0
Exp/Cntr=0.3,0.1

Type RM Length L Ch R = 1 ,6135    ,483,483,483
BEGIN DESCRIPTION:
TRIB 4 TO EIGHTEENMILE CREEK 10.0
END DESCRIPTION:
XS GIS Cut Line= 3
        2495175.       13494225.        2495975.       13493525.
      2496574.97     13493175.02
#Sta/Elev= 30
  3928.2  193.58  3985.6  192.94  4165.5  192.03  4211.5  191.89  4275.6  189.71
  4403.2  187.41  4473.5  184.67  4481.1  185.37    4538  184.03  4665.2  177.87
  4750.6  174.98  4785.7  174.14  4863.6  174.96  4899.8  173.41  4900.3  172.91
  4912.8  173.41  5063.6  174.07  5072.3  174.55  5079.3   176.8    5095  177.99
  5162.1  178.71    5188  178.78  5211.2  176.28  5245.9  178.34  5304.9   179.8
    5435  185.43  5550.7  190.94  5563.4  191.39  5652.8  194.84  5685.8  195.92
#Mann= 12 ,-1 , 0
  3928.2    .035       0  3985.6     .05       0  4165.5     .07       0
  4275.6     .05       0  4899.8     .05       0  4912.8     .05       0
  5162.1      .1       0  5304.9    .035       0    5435     .07       0
  5550.7    .035       0  5563.4     .07       0  5652.8     .05       0
Bank Sta=4899.8,4912.8
XS Rating Curve= 0 ,0
Exp/Cntr=0.3,0.1

Type RM Length L Ch R = 1 ,5652    ,468,468,468
BEGIN DESCRIPTION:
TRIB 4 TO EIGHTEENMILE CREEK 9.0
END DESCRIPTION:
XS GIS Cut Line= 3
      2495574.97     13494075.01        2495975.       13493925.
      2496575.02     13493324.98
#Sta/Elev= 30
    4568  189.76  4753.3  186.12  4766.3   185.9  4859.4  184.23  4949.8  180.83
  4973.9  178.97  4980.1  177.95  4985.4  174.36  4992.6  172.41  4998.8  172.41
  5002.8  169.28  5003.3  168.78  5015.4  168.78  5015.9  169.28  5037.7  173.09
  5051.8  174.34  5116.6  176.58  5136.7  177.53  5179.1  177.71  5292.2  176.13
  5320.5  176.74  5405.4  176.66  5419.5  177.29  5447.8  176.17  5461.9  176.95
  5574.9  178.93    5657  181.25  5689.9  183.46  5813.6  190.82  5843.8  192.32
#Mann= 11 ,-1 , 0
    4568     .07       0  4753.3     .05       0  4766.3     .07       0
  4859.4     .12       0  5002.8     .05       0  5015.9     .12       0
  5116.6     .05       0  5574.9    .035       0    5657     .05       0
  5689.9     .07       0  5813.6     .05       0
Bank Sta=5002.8,5015.9
XS Rating Curve= 0 ,0
Exp/Cntr=0.3,0.1

Type RM Length L Ch R = 1 ,5184    ,471,471,471
BEGIN DESCRIPTION:
TRIB 4 TO EIGHTEENMILE CREEK 8.0
END DESCRIPTION:
XS GIS Cut Line= 3
        2496425.     13494625.04        2496375.       13494125.
      2496674.99     13493325.03
#Sta/Elev= 30
  4497.9  190.44  4785.8  182.63  4879.8  179.27  4904.7  176.87  4947.7  171.58
  4952.7  172.28  4983.8  169.72  4984.3  169.22    4997  169.72  5021.8  171.21
  5040.5  174.73  5074.1  174.68  5212.6  175.48  5256.8  174.48  5271.9  175.59
  5278.1  177.89  5288.8  179.59  5302.1  179.75  5316.8  176.66  5320.8  175.81
  5327.1   172.8  5332.4  173.64  5342.2  171.96  5412.5  171.89    5421  173.31
  5442.8   177.2  5525.2  181.29  5643.9  185.51  5809.4     194  5854.8  194.74
#Mann= 10 ,-1 , 0
  4497.9     .05       0  4785.8     .07       0  4904.7     .12       0
  4983.8     .05       0    4997     .12       0  5074.1     .05       0
  5212.6     .07       0  5316.8     .05       0    5421     .12       0
  5525.2     .05       0
Bank Sta=4983.8,4997
XS Rating Curve= 0 ,0
Exp/Cntr=0.3,0.1

Type RM Length L Ch R = 1 ,4713    ,506,506,506
BEGIN DESCRIPTION:
TRIB 4 TO EIGHTEENMILE CREEK 7.0
END DESCRIPTION:
XS GIS Cut Line= 3
      2496474.98     13494525.04        2496775.       13494025.
      2497025.02     13493524.96
#Sta/Elev= 30
  4424.2  187.32  4540.9  183.69  4554.5  183.75  4576.4  182.59  4585.6  182.51
  4680.8   177.4  4692.5  175.95  4715.8  174.53  4768.4  174.13    4846  174.68
  4882.9  174.23  4935.4  172.59  4941.3   173.1  4972.4  170.99    4984  167.42
  4992.5  166.26    4993  165.76  5006.1  165.76  5006.6  166.26  5007.3  168.28
  5010.1  168.28  5015.7   170.8  5029.7  171.73    5066  172.68  5096.8  174.76
  5222.6  176.78  5323.3  181.14  5373.5  184.28    5432  187.11  5566.4  194.08
#Mann= 7 ,-1 , 0
  4424.2     .05       0  4576.4     .07       0  4768.4     .12       0
  4992.5     .05       0  5006.6     .12       0  5323.3     .12       0
    5432     .05       0
Bank Sta=4992.5,5006.6
XS Rating Curve= 0 ,0
Exp/Cntr=0.3,0.1

Type RM Length L Ch R = 1 ,4207    ,461,461,461
BEGIN DESCRIPTION:
TRIB 4 TO EIGHTEENMILE CREEK 6.0
END DESCRIPTION:
XS GIS Cut Line= 3
        2496575.       13494725.        2497175.       13494175.
      2497274.99     13493675.04
#Sta/Elev= 30
  4201.4  189.62  4366.2  183.81  4493.5  179.61  4534.1   177.9  4682.7  173.95
    4732  173.05  4788.7  173.92    4802  173.49  4838.7   172.5  4873.8   170.3
  4902.2  170.33  4923.2  167.86  4937.3  168.41  4944.7  167.62  4951.5  168.86
  4958.9  167.76  4965.7  168.12    4966  167.32  4966.5  166.82  4979.6  166.82
  4980.1  167.32  4994.1  168.26  5035.7  168.32  5086.7   173.3  5096.9  175.01
  5188.7  176.95  5340.8   182.9  5402.9  186.23  5462.8  188.14  5525.2  190.33
#Mann= 8 ,-1 , 0
  4201.4     .05       0  4366.2     .07       0  4493.5     .12       0
    4802      .1       0    4966     .05       0  4980.1      .1       0
  5340.8     .12       0  5462.8     .05       0
Bank Sta=4966,4980.1
XS Rating Curve= 0 ,0
Exp/Cntr=0.3,0.1

Type RM Length L Ch R = 1 ,3746    ,471,471,471
BEGIN DESCRIPTION:
TRIB 4 TO EIGHTEENMILE CREEK 5.0
END DESCRIPTION:
XS GIS Cut Line= 3
      2497125.02     13494874.97        2497425.       13494425.
      2497825.02     13493874.98
#Sta/Elev= 30
  4459.7  187.81  4539.3  185.13  4598.2  181.31  4740.6  174.12  4783.3  172.95
  4914.9  173.52  4941.9  172.44  4964.4  172.67    4972  170.51    4978  170.57
    4987  168.11  4990.4  166.49  4990.9  165.99  5004.1  165.99  5004.6  166.49
  5022.5  168.84  5037.2   169.2  5078.9  166.75  5108.3  168.06    5123     167
  5158.5  169.73  5164.7  169.01    5186  169.94  5208.8  172.89  5244.3  175.19
  5332.2  177.56  5436.7  181.18  5581.3  187.35  5643.9  190.75  5680.6  191.44
#Mann= 6 ,-1 , 0
  4459.7     .07       0  4598.2     .12       0  4783.3      .1       0
  4990.4     .05       0  5004.6      .1       0  5332.2     .12       0
Bank Sta=4990.4,5004.6
XS Rating Curve= 0 ,0
Exp/Cntr=0.3,0.1

Type RM Length L Ch R = 1 ,3275    ,406,406,406
BEGIN DESCRIPTION:
TRIB 4 TO EIGHTEENMILE CREEK 4.0
END DESCRIPTION:
XS GIS Cut Line= 3
      2497274.98     13495025.02        2497825.       13494525.
      2498024.98     13494125.04
#Sta/Elev= 30
  4252.1  188.79  4344.4   185.6  4577.5  173.58  4627.5   172.1  4685.7  171.51
  4747.8  169.71  4825.5  170.94    4889  170.32  4931.6  168.46  4953.2  168.33
    4960   167.3  4967.4  167.28  4974.4  165.55  4974.9  165.05  4988.2  165.05
  4988.7  165.55  4992.1  166.31  5017.8  167.58  5026.2  169.22  5031.8  169.41
  5048.5  173.01  5165.9  176.38  5182.7  177.53    5231  179.03  5383.9  185.36
  5389.5  184.82  5420.3  186.59  5428.7  186.06  5434.3  187.16  5442.6  186.05
#Mann= 5 ,-1 , 0
  4252.1     .12       0  4685.7      .1       0  4974.4     .05       0
  4988.7      .1       0    5231     .12       0
Bank Sta=4974.4,4988.7
XS Rating Curve= 0 ,0
Exp/Cntr=0.3,0.1

Type RM Length L Ch R = 1 ,2869    ,698,698,698
BEGIN DESCRIPTION:
Mapping XS fe76969b
END DESCRIPTION:
XS GIS Cut Line= 3
      2497356.91     13495154.81      2498127.71       13494759.
      2498940.06     13494311.16
#Sta/Elev= 30
    4110  188.09  4366.7  182.33  4468.5   177.2  4488.6  175.73  4555.1  167.51
  4568.7  166.79  4627.3  167.89  4649.5  169.65  4710.4  167.47  4782.6  168.77
  4837.9  166.42  4932.3  168.64  4977.7  166.27  4978.2  165.77    4992  166.27
  5030.5  168.15  5052.4  171.22  5058.1  170.23  5085.1   171.5  5345.9  174.23
  5395.9  175.67    5449   175.6  5536.1  177.76  5552.2   177.4  5601.5  179.28
  5639.3  178.43  5780.3  179.17  5811.8   180.2  5829.8  181.32  5904.1  181.62
#Mann= 6 ,-1 , 0
    4110     .12       0  4468.5      .1       0  4977.7     .05       0
    4992      .1       0  5085.1    .045       0  5811.8      .1       0
Bank Sta=4977.7,4992
XS Rating Curve= 0 ,0
Exp/Cntr=0.3,0.1

Type RM Length L Ch R = 1 ,2171    ,860,860,860
BEGIN DESCRIPTION:
Mapping XS c5951fbb
END DESCRIPTION:
XS GIS Cut Line= 3
        2497320.     13495263.45      2497854.68     13495173.17
      2499528.07      13494881.3
#Sta/Elev= 30
  4442.4  187.22  4599.7  185.61  4708.2  183.48  4908.6  179.44  4946.6   177.4
  4987.3  166.87  4994.5  163.08    4995  162.58  5008.9  163.08    5056  167.92
    5264  168.97  5280.4  168.71  5409.9  166.12  5654.9  170.66    5787  168.88
  5820.2  164.19  5888.4  170.61  5918.9  168.61  5934.2  165.43  5993.7  169.24
  6030.5  165.79  6121.9  169.81  6162.2  169.35  6192.9  165.41  6226.9  169.49
  6331.6  172.07  6451.8  174.91  6513.1  178.63  6527.5  177.72  6683.3  184.09
#Mann= 13 ,-1 , 0
  4442.4    .035       0  4599.7     .12       0  4708.2    .035       0
  4908.6     .05       0  4994.5     .05       0  5008.9     .05       0
    5264      .1       0  5280.4     .05       0  5409.9    .035       0
    5787      .1       0  6331.6     .07       0  6513.1    .035       0
  6527.5     .05       0
Bank Sta=4994.5,5008.9
XS Rating Curve= 0 ,0
Exp/Cntr=0.3,0.1

Type RM Length L Ch R = 1 ,1311    ,914,914,914
BEGIN DESCRIPTION:
Mapping XS d1f3b6b1
END DESCRIPTION:
XS GIS Cut Line= 3
      2496839.05     13495597.89       2498451.9     13495534.29
      2499475.97     13495436.86
#Sta/Elev= 30
  3361.9  187.97    3660  180.53  4038.4  175.23    4273     175  4391.1  174.03
    4568   170.4  4638.8  167.66  4686.6   169.1  4751.5   169.4  4919.1  165.39
  4949.1  157.08  4959.1  152.08  4991.9  151.21  4992.4  150.71  5006.6  151.21
  5029.3  166.29  5089.6  164.77  5139.8  167.53  5233.8  167.01    5347  163.04
  5380.9  163.62  5421.1  160.71  5471.3  161.86  5547.9  172.88  5581.8  175.61
  5675.2  175.76    5867  176.58  5903.3  179.22  5990.5  180.45  6004.7  181.03
#Mann= 12 ,-1 , 0
  3361.9     .05       0    3660     .12       0    4273    .035       0
  4391.1     .05       0    4568     .07       0  4686.6     .05       0
  4751.5      .1       0  4991.9     .05       0  5006.6      .1       0
    5347     .12       0  5675.2    .035       0  5990.5     .05       0
Bank Sta=4991.9,5006.6
XS Rating Curve= 0 ,0
Exp/Cntr=0.3,0.1

Type RM Length L Ch R = 1 ,397     ,0,0,0
BEGIN DESCRIPTION:
TRIB 4 TO EIGHTEENMILE CREEK 1.0
END DESCRIPTION:
XS GIS Cut Line= 3
      2496828.68     13495868.73      2498208.31     13496158.35
      2499125.04     13495624.98
#Sta/Elev= 30
  3590.3  183.21  3729.6  181.82  3817.7  178.62  3937.5  175.21  4037.4  173.82
  4291.6  172.03  4379.8  174.17  4549.4  176.18  4865.5  167.81  4910.2  162.32
  4915.3  163.23  4954.3  157.37  4960.1  158.16  4988.4  152.55  4988.9  152.05
  5003.2  152.55  5015.1  157.14  5078.7   159.3  5146.6  158.86  5181.4  162.37
  5373.4  161.46  5416.4  162.76  5437.9  161.59  5453.6  158.66  5571.1  157.54
  5678.8  167.73  5772.3   172.8  5892.2  176.92  5959.2  181.68  6060.6  183.42
#Mann= 12 ,-1 , 0
  3590.3     .05       0  3817.7    .035       0  3937.5     .07       0
  4037.4     .12       0  4379.8    .035       0  4549.4     .05       0
  4954.3      .1       0  4988.4     .05       0  5003.2      .1       0
  5078.7     .05       0  5772.3    .035       0  5959.2     .12       0
Bank Sta=4988.4,5003.2
XS Rating Curve= 0 ,0
Exp/Cntr=0.3,0.1

Chan Stop Cuts=-1
Use User Specified Reach Order=0
Composite Channel Slope=5
