--- YORKTOWN CREEK.prj (project) ---

Proj Title=YORKTOWN CREEK Base Level Engineering
Current Plan=p01
Default Exp/Contr=0.3,0.1
English Units
Geom File=g01
Flow File=f01
Plan File=p01
Y Axis Title=Elevation
X Axis Title(PF)=Main Channel Distance
X Axis Title(XS)=Station
BEGIN DESCRIPTION:
YORKTOWN CREEK
END DESCRIPTION:
DSS Export Rating Curves= 0
DSS Export Rating Curve Sorted= 0
DSS Export Volume Flow Curves= 0
DXF OffsetX= 0
DXF OffsetY= 0
DXF ScaleX= 1
DXF ScaleY= 10

--- YORKTOWN CREEK.p01 (plan) ---

Plan Title=Multiple Run
Program Version=4.10
Short Identifier=Multiple
Geom File=g01
Flow File=f01
Subcritical Flow
K Sum by GR= 0
Std Step Tol= 0.01
Critical Tol= 0.01
Num of Std Step Trials= 20
Max Error Tol= 0.3
Flow Tol Ratio= 0.001
Split Flow NTrial= 30
Split Flow Tol= 0.02
Split Flow Ratio= 0.02
Log Output Level= 0
Friction Slope Method= 1
Unsteady Friction Slope Method= 2
Unsteady Bridges Friction Slope Method= 1
Parabolic Critical Depth
Global Vel Dist= 1 , 1 , 1
Global Log Level= 0
CheckData=True
Encroach Param=-1 ,0,0, 0
BEGIN DESCRIPTION:
Multiple Run
END DESCRIPTION:
Computation Interval=1HOUR
Output Interval=1HOUR
Run HTab= 0
Run UNet= 0
Run PostProcess= 0
Run WQNet= 0
UNET Theta= 1
UNET Theta Warmup= 1
UNET ZTol= 0.02
UNET ZSATol= 0.05
UNET MxIter= 20
UNET MaxInSteps= 0
UNET DtIC= 0
UNET DtMin= 0
UNET MaxCRTS= 20
UNET WFStab= 2
UNET SFStab= 1
UNET WFX= 1
UNET SFX= 1
UNET DSS MLevel= 4
UNET DZMax Abort= 100
UNET Convert EG Bridges= 0
UNET Use Existing IB Tables=-1
UNET Froude Reduction=False
UNET Froude Limit= 1
UNET Froude Power= 10
UNET Time Slicing=0,0, 5
UNET Junction Losses=0
Instantaneous Interval=1HOUR
Write IC File= 0
Write IC File at Sim End=0
Echo Input=False
Echo Parameters=False
Echo Output=False
Write Detailed= 0
WQ AD Non Conservative
WQ ULTIMATE=-1
WQ Max Comp Step=1HOUR
WQ Output Interval=15MIN
WQ Output Selected Increments= 0
WQ Output face flow=0
WQ Output face velocity=0
WQ Output face area=0
WQ Output face dispersion=0
WQ Output cell volume=0
WQ Output cell surface area=0
WQ Output cell continuity=0
WQ Output cumulative cell continuity=0
WQ Output face conc=0
WQ Output face dconc_dx=0
WQ Output face courant=0
WQ Output face peclet=0
WQ Output face adv mass=0
WQ Output face disp mass=0
WQ Output cell mass=0
WQ Output cell source sink temp=0
WQ Output cell source sink nsm=0
WQ Output MaxMinRange=-1
WQ Daily Max Min Mean=-1
WQ Daily Range=0
WQ Daily Time=0
WQ Create Restart=0
WQ Fixed Restart=0
WQ System Summary=0
WQ Use Fixed Temperature=0
Sorting and Armoring Iterations= 10
XS Update Threshold= 0.02
Hydraulics Update Threshold= 0.02
Energy Slope Method= 1
Volume Change Method= 0
XS Weighting Method= 0
Number of US Weighted Cross Sections= 1
Number of DS Weighted Cross Sections= 1
Upstream XS Weight=0.25
Main XS Weight=0.5
Downstream XS Weight=0.25
Number of DS XS's Weighted with US Boundary= 1
Upstream Boundary Weight= 1
Weight of XSs Associated with US Boundary= 0
Number of US XS's Weighted with DS Boundary= 1
Downstream Boundary Weight= 0.5
Weight of XSs Associated with DS Boundary= 0.5
Sediment Output Level= 4
Mass or Volume Output= 0
Output Increment Type= 1
Profile and TS Output Increment= 10
XS Output Flag= 0
XS Output Increment= 10
Disregard all LS=0
Disregard all Conn=0
Disregard all Breaches=0
Disregard all Pumps=0

--- YORKTOWN CREEK.f01 (steady flow) ---

Flow Title=Multiple
Number of Profiles=7
Profile Names=10-year,25-year,50-year,1pct_min,100-year,1pct_plu,500-year
River Rch & RM= YORKTOWN CREEK,Reach-1,98695
     581     935    1253     814    1624    3240    2701
River Rch & RM= YORKTOWN CREEK,Reach-1,97020
     778    1271    1720    1127    2248    4485    3806
River Rch & RM= YORKTOWN CREEK,Reach-1,93474
     923    1518    2064    1357    2708    5403    4619
River Rch & RM= YORKTOWN CREEK,Reach-1,89217
    1005    1657    2257    1486    2964    5914    5069
River Rch & RM= YORKTOWN CREEK,Reach-1,85728
    1138    1887    2579    1702    3396    6777    5844
River Rch & RM= YORKTOWN CREEK,Reach-1,83085
    1183    1963    2686    1774    3540    7064    6101
River Rch & RM= YORKTOWN CREEK,Reach-1,81352
    1316    2195    3013    1996    3983    7948    6905
River Rch & RM= YORKTOWN CREEK,Reach-1,79896
    1385    2311    3173    2102    4194    8368    7268
River Rch & RM= YORKTOWN CREEK,Reach-1,75570
    1513    2534    3488    2316    4621    9219    8045
River Rch & RM= YORKTOWN CREEK,Reach-1,72726
    1616    2713    3739    2485    4959    9895    8654
River Rch & RM= YORKTOWN CREEK,Reach-1,65548
    1618    2714    3739    2484    4956    9889    8641
River Rch & RM= YORKTOWN CREEK,Reach-1,64806
    2778    4769    6674    4498    8975   17908   16103
River Rch & RM= YORKTOWN CREEK,Reach-1,60594
    2976    5125    7188    4854    9685   19324   17444
River Rch & RM= YORKTOWN CREEK,Reach-1,59628
    3175    5477    7690    5198   10371   20692   18714
River Rch & RM= YORKTOWN CREEK,Reach-1,52863
    4196    7305   10320    7014   13994   27921   25527
River Rch & RM= YORKTOWN CREEK,Reach-1,51759
    4874    8518   12063    8210   16381   32685   29933
River Rch & RM= YORKTOWN CREEK,Reach-1,44817
    5864   10302   14643    9998   19948   39802   36681
River Rch & RM= YORKTOWN CREEK,Reach-1,42221
    5931   10421   14814   10115   20183   40270   37119
River Rch & RM= YORKTOWN CREEK,Reach-1,41721
    5954   10459   14865   10148   20248   40400   37222
River Rch & RM= YORKTOWN CREEK,Reach-1,39309
    6118   10750   15279   10431   20813   41527   38260
River Rch & RM= YORKTOWN CREEK,Reach-1,35718
    6092   10695   15194   10368   20686   41275   37988
River Rch & RM= YORKTOWN CREEK,Reach-1,32863
    6112   10720   15219   10377   20704   41310   37962
River Rch & RM= YORKTOWN CREEK,Reach-1,29019
    6316   11085   15746   10740   21430   42758   39325
River Rch & RM= YORKTOWN CREEK,Reach-1,26590
    6287   11025   15650   10668   21285   42468   39004
River Rch & RM= YORKTOWN CREEK,Reach-1,25341
    6432   11281   16017   10919   21787   43471   39935
River Rch & RM= YORKTOWN CREEK,Reach-1,20258
    6445   11301   16041   10932   21813   43523   39959
River Rch & RM= YORKTOWN CREEK,Reach-1,16462
    6567   11515   16346   11141   22229   44353   40723
River Rch & RM= YORKTOWN CREEK,Reach-1,13990
    6590   11553   16397   11173   22292   44479   40819
River Rch & RM= YORKTOWN CREEK,Reach-1,12111
    6569   11504   16316   11110   22167   44230   40533
River Rch & RM= YORKTOWN CREEK,Reach-1,8907
    7795   13708   19499   13312   26560   52995   48808
Boundary for River Rch & Prof#=YORKTOWN CREEK,Reach-1,1
Up Type=0
Dn Type=3
Dn Slope=0.002
Boundary for River Rch & Prof#=YORKTOWN CREEK,Reach-1,2
Up Type=0
Dn Type=3
Dn Slope=0.002
Boundary for River Rch & Prof#=YORKTOWN CREEK,Reach-1,3
Up Type=0
Dn Type=3
Dn Slope=0.002
Boundary for River Rch & Prof#=YORKTOWN CREEK,Reach-1,4
Up Type=0
Dn Type=3
Dn Slope=0.002
Boundary for River Rch & Prof#=YORKTOWN CREEK,Reach-1,5
Up Type=0
Dn Type=3
Dn Slope=0.002
Boundary for River Rch & Prof#=YORKTOWN CREEK,Reach-1,6
Up Type=0
Dn Type=3
Dn Slope=0.002
Boundary for River Rch & Prof#=YORKTOWN CREEK,Reach-1,7
Up Type=0
Dn Type=3
Dn Slope=0.002

--- YORKTOWN CREEK.g01 (geometry) ---

Geom Title=Existing Conditions
Program Version=4.10

River Reach=YORKTOWN CREEK  ,Reach-1
Reach XY= 30
        2428875.       13574425.      2431664.59     13569535.16
      2434180.84     13568177.05      2437573.54     13567871.47
      2439168.79      13565582.8      2440563.42     13566073.61
      2440661.36     13565088.46      2442919.54     13564077.45
      2442778.31     13561676.74      2444767.68      13559474.9
      2444021.66     13554976.72       2442676.2      13554164.5
      2443177.06     13550630.85      2445273.39     13548668.97
       2445674.6     13546838.91      2444876.96     13545880.89
      2446575.06     13543305.01      2445830.46     13541772.54
      2449871.46     13538573.54      2448824.98      13537338.9
      2450335.76     13534465.32      2454569.06     13534622.74
      2457438.86     13532525.52      2458490.21      13533374.5
      2459545.18     13532624.71      2462823.45     13533171.25
       2465861.7     13528638.34      2467417.18     13529181.19
      2467671.25     13527826.55        2466725.       13527275.

Type RM Length L Ch R = 1 ,98695   ,188,188,188
BEGIN DESCRIPTION:
YORKTOWN CREEK 138.0
END DESCRIPTION:
XS GIS Cut Line= 3
      2429475.03     13574575.01        2428875.       13574325.
      2428274.97     13574825.03
#Sta/Elev= 30
  4404.5   406.2  4443.2  405.63  4458.7  405.22  4472.2  403.99  4490.7  403.99
  4496.1  402.88  4512.9  402.23    4703  398.45    4833  396.34    4892  396.14
  4915.3  394.82  4984.8  394.08  4985.1  393.58  4988.6  393.58  4988.8  394.08
  5039.9  394.08    5114  395.46  5160.6  396.19  5168.4  397.07  5182.8  397.35
  5238.5  397.74  5260.9  397.83  5267.4  397.09  5331.1  397.46  5473.4  399.77
  5604.7  401.74  5622.2  402.26  5750.3  404.42  5807.6  406.87  5835.6  407.35
#Mann= 9 ,-1 , 0
  4404.5    .013       0  4443.2    .035       0  4984.8    .035       0
  4988.8    .035       0    5114     .05       0  5238.5    .035       0
  5473.4     .05       0  5604.7    .035       0  5622.2     .05       0
Bank Sta=4984.8,4988.8
XS Rating Curve= 0 ,0
Exp/Cntr=0.3,0.1

Type RM Length L Ch R = 1 ,98507   ,334,334,334
BEGIN DESCRIPTION:
Mapping XS c01848e8
END DESCRIPTION:
XS GIS Cut Line= 3
      2429529.85     13574541.28      2428876.61     13574126.77
      2428108.07     13574072.64
#Sta/Elev= 30
  4284.1  407.04  4291.1   406.4  4306.4  406.74  4320.4  406.17  4327.6  405.34
  4342.8   405.1    4364  403.36  4538.6  399.59  4603.7  399.05  4655.4  397.55
    4813  394.77  4893.9   393.8  4937.5  393.75  4964.9  393.03  5053.7   392.5
    5054     392  5057.5     392  5057.7   392.5  5129.5  393.21  5149.3  394.14
  5340.1  395.01  5578.4  397.76  5583.4  397.58  5610.7  398.71  5630.8  398.24
  5650.8  398.48  5741.1  399.92  5761.1  401.14  5801.2  401.29  5828.2  401.82
#Mann= 4 ,-1 , 0
  4284.1    .013       0  4320.4    .035       0  5053.7    .035       0
  5057.7    .035       0
Bank Sta=5053.7,5057.7
XS Rating Curve= 0 ,0
Exp/Cntr=0.3,0.1

Type RM Length L Ch R = 1 ,98173   ,463,463,463
BEGIN DESCRIPTION:
YORKTOWN CREEK 137.0
END DESCRIPTION:
XS GIS Cut Line= 3
      2429575.02     13574475.02        2428975.       13573875.
      2428068.57     13573433.02
#Sta/Elev= 30
  4151.2  406.29  4179.5  404.47  4193.7  404.44  4377.5  400.02  4731.1  393.86
  4845.6  392.98  4872.5  393.01  4914.9  392.07  4985.6  391.51  5088.8  391.93
  5168.9  391.45  5169.1  390.95  5172.6  390.95  5172.9  391.45  5216.6  391.58
  5388.4  393.62  5441.9  394.46  5447.5  394.26  5455.9  394.71  5478.1  394.33
  5695.4  395.93  5768.5  396.93  5778.5  397.68  5791.1  397.99  5813.6   397.4
  5903.7  398.61  5920.7  399.68  5934.3  399.97  5956.5  399.54  6008.2     400
#Mann= 5 ,-1 , 0
  4151.2    .035       0  4845.6     .04       0  5168.9     .04       0
  5172.9     .04       0  5388.4    .035       0
Bank Sta=5168.9,5172.9
XS Rating Curve= 0 ,0
Exp/Cntr=0.3,0.1

Type RM Length L Ch R = 1 ,97710   ,690,690,690
BEGIN DESCRIPTION:
YORKTOWN CREEK 136.0
END DESCRIPTION:
XS GIS Cut Line= 3
      2429725.01       13573925.        2429325.       13573725.
      2428724.99     13572824.99
#Sta/Elev= 30
  4590.9  403.34  4613.3   403.5  4621.7  402.26  4627.2  402.74  4635.6  400.29
    4644  398.45  4649.6  398.83    4658  396.94  4666.4  396.13  4725.1  395.22
  4778.2  395.12  4800.5  394.32  4850.9  393.76  4912.3  393.63  4917.9  392.43
  4934.7  391.74  4940.3  390.47  4962.7   389.6  5139.1  389.74  5252.5  389.45
  5252.7  388.95  5256.2  388.95  5256.5  389.45  5370.1  390.21  5457.3  390.23
  5586.5  391.55  5831.3  397.59  5853.9  397.79  5968.1  400.99  6119.8  404.06
#Mann= 4 ,-1 , 0
  4590.9     .05       0  5139.1     .04       0  5252.5     .05       0
  5256.5     .04       0
Bank Sta=5252.5,5256.5
XS Rating Curve= 0 ,0
Exp/Cntr=0.3,0.1

Type RM Length L Ch R = 1 ,97020   ,458,458,458
BEGIN DESCRIPTION:
YORKTOWN CREEK 135.0
END DESCRIPTION:
XS GIS Cut Line= 3
      2429724.99     13573874.96        2429575.       13573375.
      2428975.01     13572825.01
#Sta/Elev= 30
  4442.5  402.83  4452.9  402.15  4484.2  395.96  4497.3  395.12  4530.3  395.09
  4563.4  394.41  4568.6  393.92  4733.9  392.17  4777.4  390.86  4881.8  388.85
  4910.8  387.43  4947.9  386.15  5004.5  385.44  5004.8  384.94  5008.6  384.94
  5008.9  385.44  5028.3  387.39  5047.6  387.63  5141.4  386.64  5169.5  385.48
  5219.4  386.83  5318.1  387.69  5424.8  390.19  5431.6  389.66  5445.7  389.68
  5459.9  391.26  5466.7  390.97  5474.1  391.62  5700.4  395.94  5778.4  398.03
#Mann= 6 ,-1 , 0
  4442.5     .04       0  4910.8      .1       0  5004.5     .05       0
  5008.9      .1       0  5047.6     .03       0  5141.4     .04       0
Bank Sta=5004.5,5008.9
XS Rating Curve= 0 ,0
Exp/Cntr=0.3,0.1

Type RM Length L Ch R = 1 ,96562   ,922,922,922
BEGIN DESCRIPTION:
YORKTOWN CREEK 134.0
END DESCRIPTION:
XS GIS Cut Line= 3
      2430274.98     13573524.98        2429675.       13572925.
        2429075.       13572675.
#Sta/Elev= 30
  4292.9  398.29  4454.4  395.29  4530.9   393.9  4567.1  393.51  4686.5  392.28
  4731.3     391  4773.7  388.15    4872  386.46  4995.5  385.42  5042.4   386.3
  5113.1  386.25  5188.8  385.19  5217.2  384.81  5238.9  383.31  5269.2  382.34
  5269.5  381.84  5273.3  381.84  5273.6  382.34  5346.6  385.16  5401.4  386.79
  5448.8  387.24  5531.4  388.18  5585.6  389.65  5617.5  391.31    5676  391.94
  5693.9  393.83  5723.7  393.71  5747.5  394.39  5782.2  396.79  5791.4  396.57
#Mann= 12 ,-1 , 0
  4292.9    .035       0  4454.4     .05       0  4530.9    .035       0
  4567.1     .05       0  4686.5     .04       0    4872      .1       0
  4995.5     .04       0  5188.8     .05       0  5269.2     .04       0
  5273.6     .05       0  5346.6     .04       0  5448.8    .035       0
Bank Sta=5269.2,5273.6
XS Rating Curve= 0 ,0
Exp/Cntr=0.3,0.1

Type RM Length L Ch R = 1 ,95640   ,455,455,455
BEGIN DESCRIPTION:
Mapping XS fbad51cc
END DESCRIPTION:
XS GIS Cut Line= 4
      2430656.46     13573344.59      2429910.72     13572703.57
      2429552.32     13572566.84       2428975.9     13572434.89
#Sta/Elev= 30
  3616.8  402.79  3986.7   394.2  4097.9  392.34  4213.7  389.71  4383.6  387.51
  4505.4  385.75    4511  385.64  4574.9  384.39  4626.3  384.35  4873.9  383.22
  4938.7  381.81  4980.7  381.75  5019.8  381.03  5020.1  380.53  5024.3  381.03
  5114.4  387.26  5149.6  388.12  5165.7  389.23  5192.5  389.07  5278.4  390.83
    5299  391.99  5331.5  392.03  5360.6  392.98  5369.3  394.15  5411.9  394.37
  5460.3  396.74  5514.5   397.1  5545.3  398.39  5551.3  399.37  5575.1  399.66
#Mann= 11 ,-1 , 0
  3616.8    .035       0  4097.9     .05       0  4213.7    .035       0
  4383.6     .05       0  4505.4      .1       0    4511     .05       0
  4626.3    .035       0  4938.7      .1       0  4980.7    .035       0
  5019.8    .035       0  5024.3    .035       0
Bank Sta=5019.8,5024.3
XS Rating Curve= 0 ,0
Exp/Cntr=0.3,0.1

Type RM Length L Ch R = 1 ,95185   ,354,354,354
BEGIN DESCRIPTION:
Mapping XS 93240fbd
END DESCRIPTION:
XS GIS Cut Line= 4
      2430739.86     13573157.15      2429962.05     13572546.01
       2429892.6     13572261.28      2429539.25     13572004.93
#Sta/Elev= 30
  3834.3  401.54  3939.4  399.81  3974.7  398.45  4024.4  397.83  4074.1  396.12
  4209.3  393.44  4266.6  391.74  4301.9  391.68  4351.6  390.35  4430.2  389.67
    4488  388.01  4558.5   387.6  4601.9  386.51  4672.4  386.26  4788.4  384.68
    4793  384.58  4826.6  383.88  4906.9  380.85  5007.5   380.2  5007.8   379.7
  5011.7   379.7  5012.1   380.2  5228.2  383.06  5290.9  383.91  5326.4  385.78
  5385.2  385.96  5434.8  388.54  5491.9  388.59  5548.3  391.56  5553.1   391.2
#Mann= 6 ,-1 , 0
  3834.3    .035       0  4788.4     .05       0    4793    .035       0
  5007.5    .035       0  5012.1    .035       0  5228.2    .035       0
Bank Sta=5007.5,5012.1
XS Rating Curve= 0 ,0
Exp/Cntr=0.3,0.1

Type RM Length L Ch R = 1 ,94831   ,594,594,594
BEGIN DESCRIPTION:
YORKTOWN CREEK 131.0
END DESCRIPTION:
XS GIS Cut Line= 3
      2430975.03     13573075.03        2430175.       13572275.
      2429625.02     13571725.02
#Sta/Elev= 30
  3869.2  406.23  3883.4  406.04  3897.5  404.21  3925.8   403.8    3941  402.28
  4095.5  399.47  4392.5  392.08  4562.2  389.68  4604.6  388.22    4746  387.39
    4892  383.95  4972.3  379.33  5012.4  379.06  5012.7  378.56  5016.7  378.56
    5017  379.06  5110.6  380.39  5144.7  380.96  5245.8  381.09  5288.2  381.18
    5381  382.17  5467.3  384.16  5509.7  386.35  5552.1  386.43  5594.6  388.85
    5637  389.16  5679.4  391.74    5712  391.88  5741.1  392.61  5778.4   394.2
#Mann= 12 ,-1 , 0
  3869.2    .013       0    3941    .035       0    4892     .05       0
  5012.4     .05       0    5017     .05       0  5110.6    .035       0
  5144.7     .05       0  5245.8    .035       0  5288.2     .05       0
    5381    .035       0    5712     .05       0  5741.1    .035       0
Bank Sta=5012.4,5017
XS Rating Curve= 0 ,0
Exp/Cntr=0.3,0.1

Type RM Length L Ch R = 1 ,94237   ,763,763,763
BEGIN DESCRIPTION:
YORKTOWN CREEK 130.0
END DESCRIPTION:
XS GIS Cut Line= 3
      2430774.99     13572424.99        2430225.       13571825.
        2429925.       13571525.
#Sta/Elev= 30
  4043.9  390.67  4093.5  390.06  4164.4   388.2    4228  387.61  4267.5   386.6
    4313  385.82    4334  386.71  4341.4  386.65  4362.4  384.94  4382.6  384.58
  4525.2  382.51  4546.1  382.97  4567.7  381.98  4641.3  380.84  4778.1  379.39
  4808.2  379.62  4914.4  378.35    4971   378.2  4996.9   377.1  4997.2   376.6
  5001.3   376.6  5001.7   377.1  5041.7  377.52  5055.8  378.19  5098.2  380.89
  5112.4  382.65    5154   384.8  5225.5   387.4  5239.7  388.31  5282.1  389.18
#Mann= 8 ,-1 , 0
  4043.9    .035       0  4267.5    .013       0  4382.6    .035       0
  4641.3     .04       0  4778.1      .1       0  4996.9     .05       0
  5001.7      .1       0    5154    .035       0
Bank Sta=4996.9,5001.7
XS Rating Curve= 0 ,0
Exp/Cntr=0.3,0.1

Type RM Length L Ch R = 1 ,93474   ,228,228,228
BEGIN DESCRIPTION:
Mapping XS 1c564177
END DESCRIPTION:
XS GIS Cut Line= 3
      2430989.81     13572309.87      2430614.82     13571351.56
       2430191.2     13570775.15
#Sta/Elev= 30
  3958.8  391.15  4237.4  385.79  4292.7  386.36  4319.4  384.61  4368.3  383.55
  4436.5  383.41  4452.4  382.46  4506.7  381.26  4720.9  378.64  4740.3  378.57
  4836.1  377.61  4886.7  377.71  4898.3  376.83  5013.9  375.73  5043.1     376
  5046.8  375.44  5047.2  374.94  5051.4  374.94  5051.8  375.44  5084.8  376.77
  5128.7  377.16  5149.6  378.48    5176   378.8  5279.2  379.34  5429.6  383.33
    5486  385.45  5600.9  387.93  5636.4  388.08  5665.7  389.14  5703.2  389.37
#Mann= 10 ,-1 , 0
  3958.8    .035       0  4237.4    .013       0  4292.7     .04       0
  4720.9     .05       0  4740.3     .04       0  4836.1     .05       0
  5013.9     .04       0  5046.8     .05       0  5051.8     .04       0
    5176     .04       0
Bank Sta=5046.8,5051.8
XS Rating Curve= 0 ,0
Exp/Cntr=0.3,0.1

Type RM Length L Ch R = 1 ,93246   ,684,684,684
BEGIN DESCRIPTION:
Mapping XS 32e0cfda
END DESCRIPTION:
XS GIS Cut Line= 3
      2431205.11     13572164.08      2430774.55     13571177.95
      2430434.26     13570400.16
#Sta/Elev= 30
  3975.8  391.91  4034.4  390.58  4038.7  390.46  4415.1  383.05  4618.7  379.82
  4759.1  378.52  4811.4   377.2    4910  376.31  4933.9  375.96    4957   374.6
  5018.9  374.72    5033  375.09  5067.3   374.4  5114.1  375.74  5127.8   374.3
    5129  374.14  5129.3  373.64  5133.6  373.64    5134  374.14  5142.9  375.47
  5187.4  375.92  5236.7  376.37  5417.7  378.71  5454.6  379.18    5648  382.65
  5672.5   383.1  5812.6  385.26  5878.3  385.58  5890.4  385.78  5900.8  385.78
#Mann= 17 ,-1 , 0
  3975.8     .04       0  4034.4    .013       0  4038.7     .04       0
    4910     .05       0    4957    .013       0  5018.9     .05       0
  5127.8     .04       0    5129     .03       0    5134     .04       0
  5187.4    .013       0  5236.7     .04       0  5417.7    .013       0
  5454.6     .04       0    5648    .013       0  5672.5     .04       0
  5878.3    .013       0  5890.4     .04       0
Bank Sta=5129,5134
XS Rating Curve= 0 ,0
Exp/Cntr=0.3,0.1

Type RM Length L Ch R = 1 ,92562   ,912,912,912
BEGIN DESCRIPTION:
Mapping XS dda91555
END DESCRIPTION:
XS GIS Cut Line= 3
      2431302.32     13572011.25       2431205.1     13570927.95
      2430510.65     13570212.66
#Sta/Elev= 30
  3853.6  390.79  4120.9  385.44    4402  380.99  4602.9  379.11  4673.1  377.26
  4852.4  375.63  4934.2  374.48  4957.6  373.71  4978.8  371.75  5004.5   371.6
  5004.9   371.1  5009.2   371.1  5009.6   371.6  5042.5  371.61  5049.5  372.37
  5063.8  372.53  5084.7  372.81  5098.9  374.22  5148.5  374.01  5162.7  372.12
  5169.6  372.18  5176.8  373.55  5183.8   373.9  5205.1  373.44  5233.4  374.14
  5261.7  373.74    5389  374.99  5516.3  377.13  5756.6  382.75  5938.2   384.4
#Mann= 5 ,-1 , 0
  3853.6     .04       0  4852.4     .05       0  5004.5     .05       0
  5009.6     .05       0  5063.8     .04       0
Bank Sta=5004.5,5009.6
XS Rating Curve= 0 ,0
Exp/Cntr=0.3,0.1

Type RM Length L Ch R = 1 ,91650   ,980,980,980
BEGIN DESCRIPTION:
Mapping XS 7876b7cf
END DESCRIPTION:
XS GIS Cut Line= 3
      2432066.22     13571171.02      2431338.95     13570274.76
      2430518.78     13569782.82
#Sta/Elev= 30
  3543.9  388.72  3588.3  385.93  3741.3  382.27  3747.7  384.37  3790.9  384.32
  3797.3  381.95  3812.1  381.21  3939.5   376.8  4104.1  374.37  4508.5  372.27
  4558.1  368.24  4586.8  371.41  4615.6  370.54  4636.4  371.83  4737.7  369.62
  4962.6  369.37  4981.4  367.14  4981.8  366.64  4986.6  367.14  4999.5  368.31
  5057.8  381.33  5079.2  382.23  5110.3  382.01  5116.2   378.8  5122.5  380.71
  5131.7  380.91  5137.5  378.87  5145.8  379.86    5190  377.07  5654.5  380.48
#Mann= 5 ,-1 , 0
  3543.9     .04       0  3588.3    .013       0  3812.1     .04       0
  4981.4     .04       0  4986.6     .04       0
Bank Sta=4981.4,4986.6
XS Rating Curve= 0 ,0
Exp/Cntr=0.3,0.1

Type RM Length L Ch R = 1 ,90670   ,1453,1453,1453
BEGIN DESCRIPTION:
Mapping XS 6946c4b7
END DESCRIPTION:
XS GIS Cut Line= 3
      2431878.72      13570726.6      2431837.05     13570018.23
      2431170.72     13569379.67
#Sta/Elev= 30
    4075  375.63  4437.2  371.24  4507.3  371.43  4687.7  369.81  4789.5  369.68
  4833.1   366.2  4833.5   365.7  4838.8   366.2  4844.8  366.27    4859  368.98
  4873.1  370.44  4887.3  370.33  4901.4  369.14  4922.8  369.73  4972.2  367.28
  5014.6  366.23  5021.9  367.01  5071.2  367.15  5134.8  368.26  5156.1  369.33
  5262.1  370.93  5396.7  374.98  5417.8  374.35  5481.3  376.97  5502.7  376.57
  5566.2     379  5587.6  378.82  5644.2  381.23  5672.5  381.23  5707.5  382.45
#Mann= 3 ,-1 , 0
    4075     .04       0  4833.1     .04       0  4838.8     .04       0
Bank Sta=4833.1,4838.8
XS Rating Curve= 0 ,0
Exp/Cntr=0.3,0.1

Type RM Length L Ch R = 1 ,89217   ,692,692,692
BEGIN DESCRIPTION:
Mapping XS 4e690654
END DESCRIPTION:
XS GIS Cut Line= 4
      2431996.76     13570525.19      2432371.77     13569733.51
       2432767.6     13568761.28      2432760.66     13568462.69
#Sta/Elev= 30
  3693.6  374.27    3865  373.12  3978.7   370.9  4444.7  367.72  4541.2   366.3
    4564  363.61  4600.4  362.61  4718.9  365.97  4924.3  363.99  4988.9  361.67
  4989.4  361.17  4994.9  361.67  5032.3  364.27  5045.4  366.67  5160.2  368.63
  5297.2  370.42  5366.3  371.71  5385.1  373.01  5471.5  374.39  5507.3  374.66
  5517.2   376.4  5521.6  375.17  5528.9  376.67  5545.6  377.56  5619.3   377.9
  5645.6  379.54    5723  380.84  5855.7  383.52  5885.7   385.2    5918  384.98
#Mann= 9 ,-1 , 0
  3693.6     .04       0  4988.9     .04       0  4994.9     .04       0
  5160.2    .013       0  5297.2     .04       0  5366.3    .013       0
  5471.5     .04       0  5517.2    .013       0    5723     .04       0
Bank Sta=4988.9,4994.9
XS Rating Curve= 0 ,0
Exp/Cntr=0.3,0.1

Type RM Length L Ch R = 1 ,88525   ,1406,1406,1406
BEGIN DESCRIPTION:
Mapping XS c5de8e1f
END DESCRIPTION:
XS GIS Cut Line= 4
      2432239.83     13570775.16      2432691.21     13569754.34
      2433107.88     13568684.89      2432996.76     13568351.54
#Sta/Elev= 30
  3915.4  383.57    4139  381.04  4481.6  374.39  4752.1  370.79    4845  369.98
  4911.9  363.58  4921.5  362.58  4930.7  358.81  4931.2  358.31  4936.8  358.81
  4965.2  363.13  5127.4  361.57  5170.8  362.11    5190  363.82  5195.3  362.88
  5271.3  364.12  5423.2  363.97  5522.4  363.69  5690.1  363.18  6189.7  367.46
  6274.1  371.66  6299.8  371.91  6337.3   374.7  6357.7  374.77  6379.5  373.09
  6389.4  373.74  6394.6  375.93  6400.6  376.73  6426.1  377.38  6530.7  379.32
#Mann= 9 ,-1 , 0
  3915.4     .04       0  4752.1    .013       0  4911.9     .05       0
  4930.7     .05       0  4936.8     .05       0  5271.3    .013       0
  5423.2     .05       0  5522.4    .013       0  6426.1     .04       0
Bank Sta=4930.7,4936.8
XS Rating Curve= 0 ,0
Exp/Cntr=0.3,0.1

Type RM Length L Ch R = 1 ,87119   ,966,966,966
BEGIN DESCRIPTION:
Mapping XS 017f172b
END DESCRIPTION:
XS GIS Cut Line= 4
       2433911.7     13570353.29      2433666.91     13569202.26
      2433255.45     13568806.42      2433052.33     13568046.01
#Sta/Elev= 30
  3598.1  384.91  3886.5  380.34    4372  367.54  4684.4   363.7  4715.3  363.47
  4763.5  363.84  4915.9  361.97  4972.2  356.74  4983.1  354.12  4983.6  353.62
  4989.5  354.12  5000.5  357.72  5048.3  357.98  5135.1  358.18    5142  357.01
  5149.2  358.18  5184.4  360.21  5236.8   361.5  5439.4  363.61  5542.2  366.27
  5699.2   370.7  5755.3  373.27  5771.7  372.69  5795.4  375.05  5830.3  375.02
  5844.1  373.98  5864.8  374.67  5875.5  376.48  5895.4  376.65  6132.9  378.78
#Mann= 12 ,-1 , 0
  3598.1    .035       0  3886.5     .04       0    4372     .05       0
  4684.4     .04       0  4715.3     .05       0  4983.1     .05       0
  4989.5     .05       0  5048.3      .1       0  5236.8     .05       0
  5439.4     .12       0  5542.2    .013       0  5895.4    .035       0
Bank Sta=4983.1,4989.5
XS Rating Curve= 0 ,0
Exp/Cntr=0.3,0.1

Type RM Length L Ch R = 1 ,86153   ,425,425,425
BEGIN DESCRIPTION:
Mapping XS a628ed4b
END DESCRIPTION:
XS GIS Cut Line= 3
       2434979.4     13570040.78      2433995.03     13568530.38
      2433265.89     13567775.19
#Sta/Elev= 30
  3190.8  374.87  3610.2  369.99  3639.3  371.11    3646  369.52  3718.9  367.57
  3746.8  368.41  3782.6  366.45  3884.9  366.15  3905.9  364.34  4421.3   360.2
  4874.7  359.48  4932.4  357.87  4983.4  354.68  4993.7  355.75  5001.2  352.91
  5001.7  352.41  5007.7  352.91  5018.6  355.51    5040  357.21  5147.1  358.45
  5655.6  369.51  5683.4  372.32  5704.7  371.77  5711.7  369.76  5725.8  371.72
  5874.5  372.33  5902.8  375.95  5938.1  373.69  5996.4   374.2  6043.4  374.56
#Mann= 9 ,-1 , 0
  3190.8    .035       0    3646     .04       0  4421.3     .05       0
  4932.4      .1       0  5001.2     .05       0  5007.7      .1       0
  5147.1     .12       0  5655.6    .013       0  5996.4    .035       0
Bank Sta=5001.2,5007.7
XS Rating Curve= 0 ,0
Exp/Cntr=0.3,0.1

Type RM Length L Ch R = 1 ,85728   ,570,570,570
BEGIN DESCRIPTION:
Mapping XS ce5be014
END DESCRIPTION:
XS GIS Cut Line= 3
      2435041.89      13570061.6       2434349.2      13568540.8
      2433855.02     13567588.85
#Sta/Elev= 30
  2928.8  375.12  3363.4  369.45  3391.9  369.47  3410.6  370.63  3430.5  368.04
  3518.4  367.26  3541.2  365.97  3639.3  364.54  3656.5  365.34  3679.5  364.01
  3869.4  361.35  4185.8  358.59  4473.2  357.97  4507.4  357.23    4599  358.09
  4606.5  357.43  4638.1  358.15  4835.5  357.84  4969.9  354.82  4988.5  351.86
    4989  351.36  4995.5  351.86  5000.8  351.93  5014.1  354.56  5030.6  359.78
  5052.7  362.76  5144.6  365.32  5507.8  371.81  5622.2  374.27  5672.5  374.51
#Mann= 8 ,-1 , 0
  2928.8    .035       0  3410.6     .04       0  4185.8     .05       0
  4835.5     .12       0  4988.5     .05       0  4995.5     .12       0
  5144.6     .05       0  5507.8    .013       0
Bank Sta=4988.5,4995.5
XS Rating Curve= 0 ,0
Exp/Cntr=0.3,0.1

Type RM Length L Ch R = 1 ,85158   ,291,291,291
BEGIN DESCRIPTION:
Mapping XS 66dab83e
END DESCRIPTION:
XS GIS Cut Line= 4
      2435187.72     13570066.79       2434661.7     13568655.38
      2434713.78     13567905.38      2434334.62     13567318.46
#Sta/Elev= 30
  3161.6  375.42  3590.4  369.39  3686.4  368.39  3707.8  369.42  3731.1  366.77
  3784.2  365.86  3816.8  366.39  3835.8  365.06  3927.4  363.38  3952.4  364.46
  3974.6  363.04  4482.9  357.54  4508.2  358.62  4518.8  357.81  4642.8  356.35
  4665.4  357.05  4893.1  356.52  4948.9  355.68    4989  352.24  4995.5  350.86
    4996  350.36  5002.6  350.86  5029.1   354.2  5080.3  353.81  5129.3  357.23
  5209.5  359.67  5270.9  360.16  5535.2  367.07  5729.6     371  6118.4   375.9
#Mann= 8 ,-1 , 0
  3161.6    .035       0  3784.2     .04       0  4482.9     .05       0
  4893.1      .1       0  4995.5     .05       0  5002.6      .1       0
  5129.3     .12       0  5270.9    .035       0
Bank Sta=4995.5,5002.6
XS Rating Curve= 0 ,0
Exp/Cntr=0.3,0.1

Type RM Length L Ch R = 1 ,84867   ,588,588,588
BEGIN DESCRIPTION:
Mapping XS 17ba69c6
END DESCRIPTION:
XS GIS Cut Line= 4
      2435489.81     13570113.68      2434937.74     13568775.17
      2434948.16     13567926.21      2434474.18     13567160.56
#Sta/Elev= 30
  3101.2  376.49  3770.4  367.49  3802.9  368.27  3832.5  365.41  3877.7  364.42
  3921.9   364.9    3939  363.55  3986.8  362.89  4051.7  363.17  4084.1  361.42
  4509.5  357.04  4559.3  357.35  4786.7  354.31  4809.3  353.85  4869.3  355.64
  4929.3  353.18  4953.3  353.65  4969.3  352.84  4979.3  350.53  4995.7  350.08
  4996.2  349.58  5002.8  350.08  5009.3  351.79  5051.8  354.62  5089.3  356.71
    5156  357.24  5285.8  359.28    5699  369.36    5917  373.04  6298.6  377.15
#Mann= 10 ,-1 , 0
  3101.2    .035       0  3877.7     .04       0  4509.5     .05       0
  4786.7      .1       0  4953.3     .12       0  4995.7     .05       0
  5002.8     .12       0  5051.8     .05       0    5156     .12       0
  5285.8    .035       0
Bank Sta=4995.7,5002.8
XS Rating Curve= 0 ,0
Exp/Cntr=0.3,0.1

Type RM Length L Ch R = 1 ,84279   ,185,185,185
BEGIN DESCRIPTION:
Mapping XS 14cae11e
END DESCRIPTION:
XS GIS Cut Line= 3
      2436156.48     13570139.73      2435432.53     13568530.38
      2434656.49     13567040.79
#Sta/Elev= 30
  3223.6  375.42  3224.9  375.42    3398     375  3450.3  374.47  3484.8  375.08
  3727.3  372.64  4114.2   366.1  4240.9     366  4273.9  363.74  4351.9  361.77
  4460.3  361.24  4492.8  359.86  4577.2  358.94  4602.3  358.77  4711.8  357.75
  4802.6  356.65  4847.2  356.74  4905.7   354.8  4950.8  352.65  4970.1  349.37
  4970.6  348.87  4977.7  349.37  4991.2  352.03  5041.8  352.18  5154.6  354.08
  5486.4  356.74  5626.4  359.09  5777.6  363.92  6101.3  370.94  6667.9  376.32
#Mann= 18 ,-1 , 0
  3223.6    .013       0  3224.9    .035       0    3398    .013       0
  3450.3    .035       0  4273.9    .013       0  4351.9    .035       0
  4492.8    .013       0  4577.2     .04       0  4602.3     .05       0
  4711.8    .013       0  4802.6     .05       0  4905.7     .12       0
  4970.1     .05       0  4977.7     .12       0  5041.8      .1       0
  5154.6     .05       0  5486.4     .12       0  5777.6    .035       0
Bank Sta=4970.1,4977.7
XS Rating Curve= 0 ,0
Exp/Cntr=0.3,0.1

Type RM Length L Ch R = 1 ,84094   ,513,513,513
BEGIN DESCRIPTION:
Mapping XS 1c0654e0
END DESCRIPTION:
XS GIS Cut Line= 3
      2436343.99     13570124.14      2435557.53     13568379.34
      2434906.96      13566968.9
#Sta/Elev= 30
  3130.6  374.81  3581.3  374.45    3749  372.68  4354.9  359.52  4664.3  356.91
  4705.5  355.98  4775.6  355.32  4884.7  351.88  4910.2  352.52  4924.6   352.9
  4950.5  352.12  4960.7  349.68  4962.4  348.22  4962.9  347.72    4970  348.22
  5012.5   351.9  5104.3  352.31  5133.6  353.79    5144  354.03  5354.7  355.44
    5364  355.45  5575.8  358.59    5584  358.62    5804  363.62    6024  368.29
  6133.9  369.41  6243.9  369.61  6353.9  370.97  6532.6  372.88  6597.7  373.53
#Mann= 20 ,-1 , 0
  3130.6     .04       0  3581.3    .035       0  4664.3    .013       0
  4705.5     .05       0  4910.2    .013       0  4924.6      .1       0
  4962.4     .05       0    4970      .1       0  5133.6    .013       0
    5144     .05       0  5354.7    .013       0    5364     .05       0
  5575.8    .013       0    5584     .05       0    5804     .04       0
    6024    .035       0  6133.9     .04       0  6243.9    .035       0
  6353.9     .04       0  6532.6    .013       0
Bank Sta=4962.4,4970
XS Rating Curve= 0 ,0
Exp/Cntr=0.3,0.1

Type RM Length L Ch R = 1 ,83581   ,496,496,496
BEGIN DESCRIPTION:
Mapping XS 2bab466a
END DESCRIPTION:
XS GIS Cut Line= 3
      2436349.21     13569191.88      2436031.49     13568316.84
      2435281.48     13567561.62
#Sta/Elev= 30
    3965  365.07  4137.9  360.22    4255  357.87    4552  354.47  4855.3  352.65
    4915  350.99  4923.6  350.77  4951.3  352.53  4972.5  350.52  4979.6   350.9
  4993.8   350.2  5000.8  348.44  5007.9  347.69  5011.1  346.43  5011.6  345.93
  5018.8  346.43  5022.1  346.72  5029.1  349.35  5043.2  350.23  5078.6  349.84
    5121  350.49  5177.6  349.45  5205.9  350.45  5241.4  350.15  5340.2  354.13
  5396.8  355.31    5418  356.64  5437.8  356.38  5707.9  359.05  5960.3  364.76
#Mann= 8 ,-1 , 0
    3965    .035       0    4552     .04       0    4915     .05       0
  4923.6      .1       0  5011.1     .05       0  5018.8      .1       0
  5241.4     .05       0  5437.8     .04       0
Bank Sta=5011.1,5018.8
XS Rating Curve= 0 ,0
Exp/Cntr=0.3,0.1

Type RM Length L Ch R = 1 ,83085   ,438,438,438
BEGIN DESCRIPTION:
Mapping XS c8b93b17
END DESCRIPTION:
XS GIS Cut Line= 3
      2436448.15     13569249.11      2436151.28     13568030.38
      2435449.09     13567224.16
#Sta/Elev= 30
  3485.2   366.7  3772.8  359.27  3911.4  356.47  4163.5  353.61  4200.2  354.03
  4278.5   352.6  4320.2  352.89  4518.7   351.2  4780.4  351.98    4868  351.06
  4932.4  348.48  4967.7  348.72  4981.9  349.62  4988.6  348.54  4998.8  345.35
  4999.3  344.85  5006.8  345.35  5010.4  347.44  5017.1  349.33  5024.7  350.24
  5109.2  353.84    5131  355.81  5156.3  356.25  5250.6  356.84  5463.3  360.29
  5485.1  361.34    5506  360.94  5583.9  362.27  5605.7  363.27  5808.7  365.36
#Mann= 6 ,-1 , 0
  3485.2    .035       0  4163.5     .04       0  4780.4      .1       0
  4998.8     .05       0  5006.8      .1       0  5156.3     .04       0
Bank Sta=4998.8,5006.8
XS Rating Curve= 0 ,0
Exp/Cntr=0.3,0.1

Type RM Length L Ch R = 1 ,82647   ,263,263,263
BEGIN DESCRIPTION:
Mapping XS 4f1104da
END DESCRIPTION:
XS GIS Cut Line= 3
      2436521.07      13569316.8      2436448.16     13567889.76
      2436026.27     13567092.85
#Sta/Elev= 30
  3329.4  367.99    3912  354.43  4072.2   352.7  4126.8  352.97  4282.4  351.01
    4430  350.82  4552.2  350.87  4844.2  350.73    4883  349.39  4926.6  348.95
  4948.6   347.9  4964.9  345.59  4978.7  347.65  4988.5  345.21    4989  344.71
  4996.6  345.21  5008.9  348.62  5036.6  349.39  5069.2  351.97  5080.6  353.77
  5091.2  353.13  5118.9  355.36  5174.8  356.52  5220.1  357.26  5300.9  359.22
  5376.2  360.61    5498  363.13    5520  362.44  5613.6  365.05    5660  365.19
#Mann= 11 ,-1 , 0
  3329.4    .035       0  4126.8     .04       0    4430     .05       0
  4552.2     .04       0    4883      .1       0  4988.5     .05       0
  4996.6      .1       0  5174.8     .05       0  5220.1     .04       0
  5300.9     .05       0  5376.2     .04       0
Bank Sta=4988.5,4996.6
XS Rating Curve= 0 ,0
Exp/Cntr=0.3,0.1

Type RM Length L Ch R = 1 ,82384   ,379,379,379
BEGIN DESCRIPTION:
Mapping XS 7c3b3460
END DESCRIPTION:
XS GIS Cut Line= 3
      2436643.47     13569161.41      2436721.59     13567863.71
      2436148.66     13566887.12
#Sta/Elev= 30
  3422.8  364.25  3789.9  355.19  3960.2  352.71  4078.4  352.17  4359.7  350.34
  4559.4  350.45  4761.7  349.54  4814.1  350.01  4877.9  348.22  4939.6  346.35
  4961.1  347.11  4976.4  344.95  4988.4  344.81  4994.2  343.17  4994.7  342.67
  5002.3  343.17  5011.2  343.71  5019.7  347.03  5025.5  346.73  5041.2  350.01
  5146.7  355.23  5327.1  357.51  5473.1  359.97  5478.9  360.69    5516  360.54
    5559  362.15  5639.1  362.93  5654.7   363.8  5676.2  363.53  5855.1  366.46
#Mann= 9 ,-1 , 0
  3422.8    .035       0  4078.4     .05       0  4559.4     .04       0
  4761.7     .05       0  4877.9      .1       0  4994.2     .05       0
  5002.3      .1       0  5146.7     .05       0  5327.1     .04       0
Bank Sta=4994.2,5002.3
XS Rating Curve= 0 ,0
Exp/Cntr=0.3,0.1

Type RM Length L Ch R = 1 ,82005   ,653,653,653
BEGIN DESCRIPTION:
Mapping XS 1b68222d
END DESCRIPTION:
XS GIS Cut Line= 3
      2437511.54     13569026.94      2437038.44     13567828.99
      2436674.15     13566879.24
#Sta/Elev= 30
  3493.5  361.08  3947.2  354.49  4265.7  352.29    4388  350.63  4424.5  351.22
  4549.2  349.77  4586.8  350.18  4749.1  346.83  4868.1  347.45  4876.4   347.4
  4957.1  346.84  4967.5  343.18  4989.3  344.41  4993.5  342.29    4994  341.79
  5001.6  342.29  5010.7  345.05  5021.4  345.86  5057.6  345.93  5100.4  349.43
  5112.3  349.77  5142.3  352.87  5232.1  354.71  5281.8  355.43  5306.4  352.52
  5421.2  352.93  5567.6  354.25  5578.3  355.68  5615.3  356.17  5798.7  357.73
#Mann= 8 ,-1 , 0
  3493.5    .035       0  4265.7     .05       0  4868.1     .04       0
  4876.4      .1       0  4993.5     .05       0  5001.6      .1       0
  5100.4     .05       0  5232.1     .04       0
Bank Sta=4993.5,5001.6
XS Rating Curve= 0 ,0
Exp/Cntr=0.3,0.1

Type RM Length L Ch R = 1 ,81352   ,711,711,711
BEGIN DESCRIPTION:
Mapping XS 16037261
END DESCRIPTION:
XS GIS Cut Line= 4
      2437915.17     13568957.47      2437511.53     13567989.58
      2437398.68     13567230.03      2437129.78     13566752.96
#Sta/Elev= 30
  3835.7  366.31  4053.3  364.69  4477.9   355.5  4658.3  352.81  4838.5  351.31
  4889.2  350.19  4915.2  348.72  4939.6  347.27  4949.7  345.75  4963.8  345.23
    4980  343.32  4985.5  341.39    4986  340.89  4994.2  340.89  4994.7  341.39
  5010.3  343.72  5050.8  345.55  5091.2  345.05  5136.9  346.38  5349.6  346.39
  5517.2  347.03  5616.9  347.69  5642.7  347.27  5672.6     348  5694.3  347.24
  5775.2  349.75  5791.1  350.94    5872  350.95  6102.1  353.01  6199.9  353.52
#Mann= 9 ,-1 , 0
  3835.7    .035       0  4658.3     .05       0  4915.2      .1       0
  4985.5     .05       0  4994.7      .1       0  5136.9     .05       0
  5349.6     .04       0  5517.2     .05       0  6102.1     .04       0
Bank Sta=4985.5,4994.7
XS Rating Curve= 0 ,0
Exp/Cntr=0.3,0.1

Type RM Length L Ch R = 1 ,80641   ,745,745,745
BEGIN DESCRIPTION:
Mapping XS 52325632
END DESCRIPTION:
XS GIS Cut Line= 4
      2438344.86     13568527.77      2437923.85     13567381.94
      2437472.46     13567199.65      2437177.34     13566665.83
#Sta/Elev= 30
  3624.3  363.56  3924.3  362.33  4141.9  359.43  4233.7  357.59  4360.1   354.4
  4476.9  349.81  4559.1  347.76  4604.9     347    4862  344.72  4919.3  344.81
  4967.9   342.7  4986.6  342.67  5000.7  338.11  5001.2  337.61    5010  338.11
  5010.7  341.07  5016.3  342.82  5034.8  343.83  5088.5  342.42    5135  344.19
  5147.6  343.32    5220  344.15  5242.8  342.91  5249.5  344.04  5254.9  343.37
  5291.7  345.23  5415.5  348.26  5486.5  351.27  5785.4   353.3  5941.8  355.65
#Mann= 12 ,-1 , 0
  3624.3    .035       0  4141.9     .05       0  4233.7     .12       0
  4476.9     .05       0  4559.1     .12       0  4604.9     .05       0
    4862      .1       0  4967.9     .12       0  5000.7     .05       0
    5010     .12       0  5291.7     .05       0  5785.4     .04       0
Bank Sta=5000.7,5010
XS Rating Curve= 0 ,0
Exp/Cntr=0.3,0.1

Type RM Length L Ch R = 1 ,79896   ,502,502,502
BEGIN DESCRIPTION:
Mapping XS 21bbee40
END DESCRIPTION:
XS GIS Cut Line= 3
      2438488.08     13568245.64        2438015.     13567026.04
      2437377.79     13566419.17
#Sta/Elev= 30
  3345.1  360.54  3649.9  359.32  3710.5  360.32  3774.8  358.65    3931  358.19
  4031.4  353.08  4167.8  348.31  4514.9  343.99  4524.5  340.32  4547.1  337.46
  4600.7  339.34  4614.3  337.96  4651.1  345.41  4682.1  347.75  4696.3  347.61
  4738.8  342.73    4868  342.24    4917  341.52  4972.1  341.68  4993.5  337.84
  5009.7  337.31  5010.2  336.81  5019.5  337.31  5021.8  339.98  5028.8  341.52
  5092.6  349.18  5212.8  351.09  5310.1  355.06  5445.9  358.76  5533.2  361.07
#Mann= 10 ,-1 , 0
  3345.1    .035       0  3649.9     .05       0    3931     .12       0
  4031.4     .05       0    4868      .1       0    4917     .12       0
  5009.7     .05       0  5019.5     .12       0  5310.1    .035       0
  5445.9    .013       0
Bank Sta=5009.7,5019.5
XS Rating Curve= 0 ,0
Exp/Cntr=0.3,0.1

Type RM Length L Ch R = 1 ,79394   ,377,377,377
BEGIN DESCRIPTION:
Mapping XS 7bd2df01
END DESCRIPTION:
XS GIS Cut Line= 4
      2438709.44     13567833.32      2438236.35     13566843.75
      2438106.14     13566444.44      2437846.28      13566089.3
#Sta/Elev= 30
    3813  360.59  3859.5  362.76  3927.6  360.33  3972.9  360.06  3978.5  361.23
  3995.6  359.98  4091.8  358.69  4137.2  356.97  4205.2  352.13  4341.3  347.24
  4505.6  344.39  4631.4  344.62  4653.5  343.01  4856.8  342.59  4910.4  339.52
  5013.7  340.32    5023  338.17  5028.3  338.47  5029.8  337.18  5030.3  336.68
  5039.6  337.18  5045.3  339.85  5054.9  341.49  5071.4  342.47    5176  340.99
  5300.1  344.91    5381  347.15    5459  350.09  5612.5  353.45  5769.9  357.27
#Mann= 9 ,-1 , 0
    3813     .05       0  4910.4     .12       0  5029.8     .05       0
  5039.6     .12       0  5071.4      .1       0    5176     .05       0
  5300.1     .12       0    5381     .05       0  5612.5    .035       0
Bank Sta=5029.8,5039.6
XS Rating Curve= 0 ,0
Exp/Cntr=0.3,0.1

Type RM Length L Ch R = 1 ,79017   ,424,424,424
BEGIN DESCRIPTION:
Mapping XS 23d0a07a
END DESCRIPTION:
XS GIS Cut Line= 3
      2438939.47     13567807.28      2438514.13     13566769.96
      2438059.18     13565977.05
#Sta/Elev= 30
  3928.9  353.67  3985.5  352.58  4009.5  353.36  4017.8     353  4028.1  351.53
  4057.5  350.75  4417.7  345.31  4579.8  343.89    4917  342.79  4947.3  341.91
  4954.1  341.01  4968.9  338.17  4973.1  335.33  4973.6  334.83  4982.5  334.83
    4983  335.33  4990.6  337.84  5012.9  339.31  5044.6  340.28  5124.9  340.14
  5171.1  341.09  5295.8   340.6  5332.5     342    5367  341.69  5390.1  342.85
  5435.3  342.75  5676.9   347.1  5687.3  347.76  5890.5  350.53  5964.2  351.87
#Mann= 6 ,-1 , 0
  3928.9     .05       0    4917     .12       0  4973.1     .05       0
    4983     .12       0  5687.3     .05       0  5890.5    .035       0
Bank Sta=4973.1,4983
XS Rating Curve= 0 ,0
Exp/Cntr=0.3,0.1

Type RM Length L Ch R = 1 ,78593   ,404,404,404
BEGIN DESCRIPTION:
Mapping XS fecba34b
END DESCRIPTION:
XS GIS Cut Line= 3
       2438887.4     13567408.02      2438761.53     13566557.29
      2438219.92     13565760.05
#Sta/Elev= 30
  4054.5  345.53  4097.2  345.01  4312.7  343.07    4899  341.08  4929.1  340.36
  4941.4   339.2  4965.1  339.39  4977.7  338.71  4992.1  337.06  4996.1  335.07
  4996.6  334.57  5005.5  334.57    5006  335.07    5014   337.8    5043  339.33
  5093.9   338.8  5144.7  340.31  5207.7  340.79  5252.5  342.43  5303.4     343
  5330.4  344.32  5375.2  345.14  5388.7  344.44  5432.2  344.71  5453.1  345.06
    5483  346.68    5525  347.44    5546  346.58  5562.9  347.68  5878.3  350.15
#Mann= 6 ,-1 , 0
  4054.5     .05       0  4097.2    .035       0    4899     .12       0
  4996.1     .05       0    5006     .12       0  5562.9    .035       0
Bank Sta=4996.1,5006
XS Rating Curve= 0 ,0
Exp/Cntr=0.3,0.1

Type RM Length L Ch R = 1 ,78189   ,1063,1063,1063
BEGIN DESCRIPTION:
Mapping XS 6744f97e
END DESCRIPTION:
XS GIS Cut Line= 3
       2438930.8     13567290.81      2438987.22     13566288.19
      2438557.55     13565611.13
#Sta/Elev= 30
  3831.5  344.52  4067.7  342.47  4725.1  339.78  4834.8  338.59  4934.2  338.65
  4962.5  337.71  4969.8   337.9  4977.8  337.34  4983.7   335.9  4993.8   335.1
  4994.3   334.6  5003.5   334.6    5004   335.1  5005.3  336.16  5014.2   337.9
    5029  338.93  5064.5  339.67  5135.6  339.93  5194.8  341.16  5230.3  342.28
  5238.7  342.14  5244.6  342.79  5265.9   342.7  5353.9  344.61  5375.1  346.23
  5384.3  345.19  5395.5  345.39  5419.8  346.48  5578.4  349.73  5637.6  351.42
#Mann= 5 ,-1 , 0
  3831.5    .035       0  4725.1     .12       0  4993.8     .05       0
    5004     .12       0  5395.5    .035       0
Bank Sta=4993.8,5004
XS Rating Curve= 0 ,0
Exp/Cntr=0.3,0.1

Type RM Length L Ch R = 1 ,77126   ,448,448,448
BEGIN DESCRIPTION:
Mapping XS 9246c0ef
END DESCRIPTION:
XS GIS Cut Line= 3
      2439777.14     13567182.25      2439534.09     13565871.53
      2438878.69     13565207.44
#Sta/Elev= 30
  3249.9  352.06  3449.5  344.36  3694.6  339.87  3945.5  338.29  4707.1  336.99
  4807.1  335.44  4834.4  337.15  4933.4  337.43  5011.2  335.71  5039.5  337.39
  5060.7  336.17  5078.9  337.07  5096.1  337.26  5112.1  334.15  5112.6  333.65
  5122.4  334.15  5124.4  335.85  5141.4  337.59  5152.7  340.63    5188  343.68
  5202.1  346.83  5233.5  348.77  5281.2  351.86  5308.2  353.05  5357.7   351.6
  5364.8  353.26    5409  355.88  5456.7  359.12    5485  358.64    5516  359.98
#Mann= 9 ,-1 , 0
  3249.9    .035       0  4807.1     .12       0  5078.9     .05       0
  5112.1     .05       0  5122.4     .05       0  5141.4     .12       0
  5233.5     .05       0  5281.2     .12       0    5409    .035       0
Bank Sta=5112.1,5122.4
XS Rating Curve= 0 ,0
Exp/Cntr=0.3,0.1

Type RM Length L Ch R = 1 ,76678   ,458,458,458
BEGIN DESCRIPTION:
Mapping XS f66e6628
END DESCRIPTION:
XS GIS Cut Line= 3
      2439846.59     13567160.58       2439620.9     13565932.29
      2439659.96     13565090.24
#Sta/Elev= 30
  3443.4  351.34  3510.1  350.38  3652.4  344.16  3699.7  342.88  3886.3  339.69
  4120.1  338.04  4478.5  338.05  4679.3  337.34  4719.6  337.79  4749.6  336.99
  4873.9  335.98  4919.8  335.76  4939.8  334.99  4949.8  335.67  4969.8  335.27
  4974.7  331.74  4975.2  331.24  4984.5  331.24    4985  331.74  4989.9  334.08
  5009.9  333.88  5049.9  335.72  5099.7  336.43  5104.7   335.8    5160  339.29
  5180.1  339.44  5220.1  342.64  5230.1  342.34  5272.8  343.94  5535.2  351.54
#Mann= 5 ,-1 , 0
  3443.4    .035       0  4873.9     .12       0  4974.7     .05       0
    4985     .12       0  5272.8    .035       0
Bank Sta=4974.7,4985
XS Rating Curve= 0 ,0
Exp/Cntr=0.3,0.1

Type RM Length L Ch R = 1 ,76220   ,650,650,650
BEGIN DESCRIPTION:
Mapping XS 7e09a6ca
END DESCRIPTION:
XS GIS Cut Line= 4
      2440080.98     13567321.21      2439820.55     13566049.48
      2440028.89      13565394.1      2439863.94     13565012.11
#Sta/Elev= 30
  3600.2  347.07  3831.1  349.36  4052.1  342.99  4208.8  339.98  4382.3  338.16
  4443.6  338.91    4592  337.03  4630.5  337.07  4688.5  336.35    4760   337.2
    4924     337  5046.6  335.73  5090.6  335.78  5128.1  334.78  5133.9  333.86
  5192.6   333.2  5289.3  335.19  5343.7  334.21  5353.8  332.12  5353.9  331.49
  5354.4  330.99  5364.2  331.49  5364.7  332.35  5396.5  337.25  5423.5  339.52
  5455.8  340.34    5461  339.48  5520.3     342    5620  344.23  6002.1  352.82
#Mann= 7 ,-1 , 0
  3600.2    .035       0    4592     .12       0  4630.5    .035       0
  5046.6     .12       0  5353.9    .035       0  5364.2     .12       0
    5620    .035       0
Bank Sta=5353.9,5364.2
XS Rating Curve= 0 ,0
Exp/Cntr=0.3,0.1

Type RM Length L Ch R = 1 ,75570   ,205,205,205
BEGIN DESCRIPTION:
Mapping XS afaad558
END DESCRIPTION:
XS GIS Cut Line= 4
       2440267.6     13567099.87      2440363.09     13566175.35
      2440306.66     13565628.47       2439976.8     13564955.71
#Sta/Elev= 30
  3919.4  347.38    4045  346.67  4232.9  342.03  4562.6  337.13  4665.3  336.69
  4778.8  335.19  4869.3  335.74  4949.7  333.99  4969.8  332.74  4975.6  331.32
  4980.6  332.25  4984.6  330.51  4985.1  330.01  4995.2  330.51    5010  333.97
  5030.1  332.45  5120.6  333.14  5321.7   332.4  5455.9  333.99  5469.3  335.72
  5491.6  336.57  5549.1  336.13  5711.9  340.72  5776.4  343.26    5782  342.54
  5814.6  345.49  5859.1  346.63  5871.9  347.94  5891.6  347.65  6147.9  353.11
#Mann= 8 ,-1 , 0
  3919.4    .035       0  4562.6     .05       0  4665.3     .12       0
  4984.6     .05       0  4995.2     .12       0  5549.1     .03       0
  5711.9     .12       0  5891.6    .035       0
Bank Sta=4984.6,4995.2
XS Rating Curve= 0 ,0
Exp/Cntr=0.3,0.1

Type RM Length L Ch R = 1 ,75365   ,276,276,276
BEGIN DESCRIPTION:
Mapping XS 1b9ba54c
END DESCRIPTION:
XS GIS Cut Line= 3
      2440692.95     13566878.48       2440580.1     13566175.35
      2440054.93     13564990.45
#Sta/Elev= 30
  4179.2  342.12  4388.7  340.55  4450.7  341.16  4618.2  337.12  4800.9  335.27
  4890.6  334.44  4946.4  334.15  5001.1  330.08    5023  331.78  5077.7  331.53
  5086.2  328.97  5086.7  328.47  5096.9  328.97  5099.5  330.79  5121.4  332.37
    5198  331.17  5242.1  332.54  5439.3  332.19  5569.9  333.69  5607.7   336.2
  5676.6  336.45  5758.3  337.69  5799.4  339.63  5804.9   340.9    5825  341.13
  5919.9  344.02  5978.8  347.23  6101.7  349.29  6152.6   351.2  6187.4  351.06
#Mann= 8 ,-1 , 0
  4179.2    .035       0  4800.9     .05       0  4890.6     .12       0
  5086.2     .05       0  5096.9     .12       0  5676.6     .03       0
    5825     .12       0  6101.7    .035       0
Bank Sta=5086.2,5096.9
XS Rating Curve= 0 ,0
Exp/Cntr=0.3,0.1
