--- KILGORE CREEK.prj (project) ---

Proj Title=KILGORE CREEK Base Level Engineering
Current Plan=p01
Default Exp/Contr=0.3,0.1
English Units
Geom File=g01
Flow File=f01
Plan File=p01
Y Axis Title=Elevation
X Axis Title(PF)=Main Channel Distance
X Axis Title(XS)=Station
BEGIN DESCRIPTION:
KILGORE CREEK
END DESCRIPTION:
DSS Export Rating Curves= 0
DSS Export Rating Curve Sorted= 0
DSS Export Volume Flow Curves= 0
DXF OffsetX= 0
DXF OffsetY= 0
DXF ScaleX= 1
DXF ScaleY= 10

--- KILGORE CREEK.p01 (plan) ---

Plan Title=Multiple Run
Program Version=4.10
Short Identifier=Multiple
Geom File=g01
Flow File=f01
Subcritical Flow
K Sum by GR= 0
Std Step Tol= 0.01
Critical Tol= 0.01
Num of Std Step Trials= 20
Max Error Tol= 0.3
Flow Tol Ratio= 0.001
Split Flow NTrial= 30
Split Flow Tol= 0.02
Split Flow Ratio= 0.02
Log Output Level= 0
Friction Slope Method= 1
Unsteady Friction Slope Method= 2
Unsteady Bridges Friction Slope Method= 1
Parabolic Critical Depth
Global Vel Dist= 1 , 1 , 1
Global Log Level= 0
CheckData=True
Encroach Param=-1 ,0,0, 0
BEGIN DESCRIPTION:
Multiple Run
END DESCRIPTION:
Computation Interval=1HOUR
Output Interval=1HOUR
Run HTab= 0
Run UNet= 0
Run PostProcess= 0
Run WQNet= 0
UNET Theta= 1
UNET Theta Warmup= 1
UNET ZTol= 0.02
UNET ZSATol= 0.05
UNET MxIter= 20
UNET MaxInSteps= 0
UNET DtIC= 0
UNET DtMin= 0
UNET MaxCRTS= 20
UNET WFStab= 2
UNET SFStab= 1
UNET WFX= 1
UNET SFX= 1
UNET DSS MLevel= 4
UNET DZMax Abort= 100
UNET Convert EG Bridges= 0
UNET Use Existing IB Tables=-1
UNET Froude Reduction=False
UNET Froude Limit= 1
UNET Froude Power= 10
UNET Time Slicing=0,0, 5
UNET Junction Losses=0
Instantaneous Interval=1HOUR
Write IC File= 0
Write IC File at Sim End=0
Echo Input=False
Echo Parameters=False
Echo Output=False
Write Detailed= 0
WQ AD Non Conservative
WQ ULTIMATE=-1
WQ Max Comp Step=1HOUR
WQ Output Interval=15MIN
WQ Output Selected Increments= 0
WQ Output face flow=0
WQ Output face velocity=0
WQ Output face area=0
WQ Output face dispersion=0
WQ Output cell volume=0
WQ Output cell surface area=0
WQ Output cell continuity=0
WQ Output cumulative cell continuity=0
WQ Output face conc=0
WQ Output face dconc_dx=0
WQ Output face courant=0
WQ Output face peclet=0
WQ Output face adv mass=0
WQ Output face disp mass=0
WQ Output cell mass=0
WQ Output cell source sink temp=0
WQ Output cell source sink nsm=0
WQ Output MaxMinRange=-1
WQ Daily Max Min Mean=-1
WQ Daily Range=0
WQ Daily Time=0
WQ Create Restart=0
WQ Fixed Restart=0
WQ System Summary=0
WQ Use Fixed Temperature=0
Sorting and Armoring Iterations= 10
XS Update Threshold= 0.02
Hydraulics Update Threshold= 0.02
Energy Slope Method= 1
Volume Change Method= 0
XS Weighting Method= 0
Number of US Weighted Cross Sections= 1
Number of DS Weighted Cross Sections= 1
Upstream XS Weight=0.25
Main XS Weight=0.5
Downstream XS Weight=0.25
Number of DS XS's Weighted with US Boundary= 1
Upstream Boundary Weight= 1
Weight of XSs Associated with US Boundary= 0
Number of US XS's Weighted with DS Boundary= 1
Downstream Boundary Weight= 0.5
Weight of XSs Associated with DS Boundary= 0.5
Sediment Output Level= 4
Mass or Volume Output= 0
Output Increment Type= 1
Profile and TS Output Increment= 10
XS Output Flag= 0
XS Output Increment= 10
Disregard all LS=0
Disregard all Conn=0
Disregard all Breaches=0
Disregard all Pumps=0

--- KILGORE CREEK.f01 (steady flow) ---

Flow Title=Multiple
Number of Profiles=7
Profile Names=10-year,25-year,50-year,1pct_min,100-year,1pct_plu,500-year
River Rch & RM= KILGORE CREEK,Reach-1,36044
     601     955    1269     816    1629    3250    2653
River Rch & RM= KILGORE CREEK,Reach-1,30685
     871    1408    1894    1232    2457    4903    4090
River Rch & RM= KILGORE CREEK,Reach-1,25418
    1638    2730    3745    2477    4943    9862    8525
River Rch & RM= KILGORE CREEK,Reach-1,18125
    1828    3057    4203    2785    5556   11086    9615
River Rch & RM= KILGORE CREEK,Reach-1,11942
    2451    4149    5751    3838    7658   15280   13448
River Rch & RM= KILGORE CREEK,Reach-1,7679
    2529    4270    5910    3937    7855   15672   13739
Boundary for River Rch & Prof#=KILGORE CREEK,Reach-1,1
Up Type=0
Dn Type=3
Dn Slope=0.005
Boundary for River Rch & Prof#=KILGORE CREEK,Reach-1,2
Up Type=0
Dn Type=3
Dn Slope=0.005
Boundary for River Rch & Prof#=KILGORE CREEK,Reach-1,3
Up Type=0
Dn Type=3
Dn Slope=0.005
Boundary for River Rch & Prof#=KILGORE CREEK,Reach-1,4
Up Type=0
Dn Type=3
Dn Slope=0.005
Boundary for River Rch & Prof#=KILGORE CREEK,Reach-1,5
Up Type=0
Dn Type=3
Dn Slope=0.005
Boundary for River Rch & Prof#=KILGORE CREEK,Reach-1,6
Up Type=0
Dn Type=3
Dn Slope=0.005
Boundary for River Rch & Prof#=KILGORE CREEK,Reach-1,7
Up Type=0
Dn Type=3
Dn Slope=0.005

--- KILGORE CREEK.g01 (geometry) ---

Geom Title=Existing Conditions
Program Version=4.10

River Reach=KILGORE CREEK   ,Reach-1
Reach XY= 30
        2510475.       13480325.      2510225.87     13477935.33
      2510471.84      13477867.4      2511121.46     13476323.54
       2511675.3     13473854.66      2511516.98     13473068.56
      2511132.07     13473025.01      2511573.81      13472064.5
      2511428.43     13471676.22      2511825.23     13471300.07
      2511524.47     13470399.88      2511824.03     13470085.29
      2511325.51     13468040.21      2512271.56     13467323.75
      2512378.74     13465426.52      2513019.17      13464777.3
      2512978.74     13464026.56      2513818.81     13462982.81
      2514904.97     13462875.04      2515569.17     13463123.23
      2516618.94     13462033.14      2517458.59      13461941.8
      2517224.51      13460609.8       2517673.8      13460064.5
      2517480.82     13459172.68      2518268.95     13458233.12
      2519317.31     13457881.48      2519501.42     13455897.82
      2520655.12     13456325.09        2520925.       13455775.

Type RM Length L Ch R = 1 ,36044   ,409,409,409
BEGIN DESCRIPTION:
KILGORE CREEK 72.0
END DESCRIPTION:
XS GIS Cut Line= 3
      2511124.98     13480424.99        2510525.       13480225.
      2509975.01       13480275.
#Sta/Elev= 30
  4367.7  234.38  4523.5  229.87  4626.1  227.17  4662.1  226.36  4694.5  226.06
    4705  225.33  4728.8  224.53  4757.7  223.59    4842  222.15  4905.3  220.43
  4968.5   219.4  5002.6  219.56  5008.2  219.19  5008.4  218.69  5011.9  218.69
  5012.2  219.19  5020.2  219.72  5040.3   219.5  5051.7  219.78  5070.4  220.51
  5088.8  220.57  5140.7  221.94  5150.8  221.64  5170.8   222.6  5241.1   224.4
  5291.3  225.22  5325.5   226.5  5522.3  230.49  5532.3  231.12  5552.4  231.09
#Mann= 10 ,-1 , 0
  4367.7     .07       0  4523.5     .12       0  4626.1     .07       0
  4662.1     .12       0  4728.8     .07       0  5008.2     .05       0
  5012.2     .07       0  5051.7     .12       0  5088.8     .07       0
  5325.5     .12       0
Bank Sta=5008.2,5012.2
XS Rating Curve= 0 ,0
Exp/Cntr=0.3,0.1

Type RM Length L Ch R = 1 ,35635   ,415,415,415
BEGIN DESCRIPTION:
KILGORE CREEK 71.0
END DESCRIPTION:
XS GIS Cut Line= 3
      2511125.01       13480175.        2510525.       13479875.
      2510075.01       13480125.
#Sta/Elev= 30
  4336.5  231.95  4369.3  231.28  4381.2  230.78  4425.9  230.15  4470.7  228.34
  4501.4   227.6  4568.5   225.3    4710  221.78  4783.7  220.23  4859.2  218.25
  4926.3  217.37  4954.2  217.21  4962.6  217.44  4970.4  217.16  4996.9  216.89
  4997.2  216.39  5000.7  216.39  5000.9  216.89  5004.5  217.14  5042.8  217.58
  5110.3  218.99  5133.2  219.11  5276.7  222.36  5302.5  222.85  5308.2   222.7
  5342.9  223.94  5405.4  225.85  5432.9  226.22  5448.9  226.87  5522.1  228.49
#Mann= 8 ,-1 , 0
  4336.5     .07       0  4369.3     .12       0    4710     .07       0
  4970.4     .12       0  4996.9     .05       0  5000.9     .12       0
  5276.7     .07       0  5342.9     .12       0
Bank Sta=4996.9,5000.9
XS Rating Curve= 0 ,0
Exp/Cntr=0.3,0.1

Type RM Length L Ch R = 1 ,35220   ,484,484,484
BEGIN DESCRIPTION:
KILGORE CREEK 70.0
END DESCRIPTION:
XS GIS Cut Line= 3
        2510975.       13479425.        2510475.       13479525.
      2510024.98     13479775.01
#Sta/Elev= 30
  4502.4  224.24    4635  221.58  4696.2  219.64  4706.4  219.77  4716.6  219.21
  4900.1  215.48  4930.7  215.32  4940.9  215.91  4979.7  212.79    4980  212.29
  4983.5  212.29  4983.7  212.79  5015.2  213.66  5020.3  214.51  5035.2  215.56
  5058.1  215.37  5079.8  216.63  5092.4  216.16  5123.3  216.37    5129  216.81
  5150.7  216.89  5195.3   218.3  5263.4  219.47  5304.6  220.43  5321.2  220.63
  5366.9  222.41  5388.7  222.33  5416.1  222.97  5432.1  223.73  5527.1  226.23
#Mann= 5 ,-1 , 0
  4502.4     .12       0  4979.7     .05       0  4983.7     .12       0
  5263.4     .07       0  5304.6     .12       0
Bank Sta=4979.7,4983.7
XS Rating Curve= 0 ,0
Exp/Cntr=0.3,0.1

Type RM Length L Ch R = 1 ,34736   ,326,326,326
BEGIN DESCRIPTION:
KILGORE CREEK 69.0
END DESCRIPTION:
XS GIS Cut Line= 3
      2510924.97     13479174.99        2510375.       13479075.
      2509924.99     13479525.01
#Sta/Elev= 30
    4441  223.09  4481.6  222.33  4584.5  219.37  4623.9  218.87  4644.2  218.04
  4691.3  216.81  4715.4  216.49    4817  214.09  4972.6  211.82  4989.8  210.93
  4995.4  210.22  4995.7  209.72  4999.2  209.72  4999.4  210.22  5028.3  210.39
  5042.4  211.77  5056.6  212.19  5212.1  214.75  5225.3  215.22  5282.8  216.36
    5297  217.22  5367.7   218.1    5396  219.17  5410.1  219.23  5452.5  220.59
  5551.5  222.82  5579.8  223.78    5594  223.85  5608.1  224.71  5636.4  224.87
#Mann= 5 ,-1 , 0
    4441     .12       0  4972.6     .05       0  4995.4     .05       0
  4999.4     .05       0  5225.3     .12       0
Bank Sta=4995.4,4999.4
XS Rating Curve= 0 ,0
Exp/Cntr=0.3,0.1

Type RM Length L Ch R = 1 ,34410   ,550,550,550
BEGIN DESCRIPTION:
Mapping XS d7baf0ca
END DESCRIPTION:
XS GIS Cut Line= 3
      2511151.89     13478918.68      2510339.43      13478741.6
      2509538.68     13479069.18
#Sta/Elev= 30
  4204.9  220.25  4241.6  220.55  4290.7  220.22  4314.3  219.62  4383.7   219.5
  4396.2  218.89  4488.3  218.56  4623.9  216.06  4711.8  213.82    4766  213.13
  4785.1  212.31  4940.8  209.97  4989.8  209.28    4994  208.32  4994.2  207.82
  4997.7  207.82    4998  208.32  5001.1  209.52  5010.3  209.94  5041.1  209.91
  5095.2  209.79  5164.9  210.72  5181.7  211.45  5266.3  212.11  5616.2  216.94
  5700.3  217.75  5771.1  217.88  5819.1  218.53  5824.5  218.97  5901.6  218.82
#Mann= 5 ,-1 , 0
  4204.9     .12       0  4940.8     .07       0    4994     .05       0
    4998     .07       0  5041.1     .05       0
Bank Sta=4994,4998
XS Rating Curve= 0 ,0
Exp/Cntr=0.3,0.1

Type RM Length L Ch R = 1 ,33860   ,287,287,287
BEGIN DESCRIPTION:
Mapping XS 6d7a017c
END DESCRIPTION:
XS GIS Cut Line= 3
      2511719.64     13478460.35      2510271.72     13478236.39
      2508974.81     13478350.98
#Sta/Elev= 30
  3538.2  218.33  3595.3  217.66  3644.1  216.26  3684.6  216.61  3835.7  214.45
  3869.7  214.17  3876.8  212.97  3897.1  214.68  3917.3  212.32  3934.7  211.69
  4099.4  209.45  4109.6  208.57  4119.7  209.64  4645.9  206.69  4982.3  206.18
  5060.3   207.3  5178.7  206.02    5179  205.52  5182.7  206.02    5241  207.46
  5268.8  210.86  5281.1     210  5291.2  207.78  5419.8  207.33    5524  208.25
  5721.9  210.47    5844  210.36  5983.9  213.14  6043.7  213.23  6305.3   215.9
#Mann= 9 ,-1 , 0
  3538.2     .07       0  3595.3     .05       0  3835.7    .035       0
  3934.7     .12       0  5178.7     .05       0  5182.7     .12       0
  5419.8      .1       0    5524     .12       0  6043.7     .05       0
Bank Sta=5178.7,5182.7
XS Rating Curve= 0 ,0
Exp/Cntr=0.3,0.1

Type RM Length L Ch R = 1 ,33573   ,461,461,461
BEGIN DESCRIPTION:
Mapping XS 9c2842d2
END DESCRIPTION:
XS GIS Cut Line= 3
      2511563.43     13478100.98      2510230.05     13477965.56
      2509168.79     13477986.37
#Sta/Elev= 30
  3653.9  217.63  3702.6  216.36  3722.7   217.1  3881.6  214.72  3885.4  214.65
  3981.6  213.55  3991.9  213.49  4014.2  212.64  4034.3  213.72  4059.5  211.44
  4104.6  211.55  4154.2  210.01  4413.4  206.03  4534.6  205.42  4657.9  204.13
  4838.4   205.4  4886.7  203.35  4886.9  202.85  4890.7  203.35  4898.7  204.26
    4959   205.4  4994.1  204.89  4999.2  203.57  5019.2  204.86  5279.2  208.72
  5568.9  211.82  5730.3  213.23  5875.2  215.42  5909.4  217.24  6055.6  219.44
#Mann= 12 ,-1 , 0
  3653.9     .05       0  3881.6    .035       0  3885.4     .05       0
  3981.6    .035       0  3991.9     .12       0  4413.4     .07       0
  4534.6     .12       0  4886.7     .05       0  4890.7     .12       0
  5568.9     .07       0  5730.3     .12       0  5875.2     .05       0
Bank Sta=4886.7,4890.7
XS Rating Curve= 0 ,0
Exp/Cntr=0.3,0.1

Type RM Length L Ch R = 1 ,33112   ,218,218,218
BEGIN DESCRIPTION:
Mapping XS 57f29c34
END DESCRIPTION:
XS GIS Cut Line= 3
      2511526.88     13477903.05      2510516.51     13477752.02
      2509418.79     13477627.16
#Sta/Elev= 30
  3961.7  220.07  4226.5  216.32  4236.6  215.26  4257.4  216.09  4266.9  215.05
    4309  213.76  4408.5  212.54  4428.7   210.3  4448.9  211.35  4509.6  208.63
  4588.3  206.63  4927.9  203.34  4964.6  202.43  4981.5  199.23  4994.9  199.18
  5000.5  200.04  5003.6  198.22  5003.8  197.72  5007.6  198.22  5025.1  203.09
  5155.9  203.76  5337.1  206.82  5508.2  211.42  5548.4  213.32  5598.8   213.5
  5679.3  216.07  5827.5  217.98  5926.1  218.36  6011.4  219.33  6088.1     219
#Mann= 7 ,-1 , 0
  3961.7     .05       0    4309    .035       0  4927.9     .12       0
  5003.6     .05       0  5007.6     .12       0  5827.5     .07       0
  5926.1     .12       0
Bank Sta=5003.6,5007.6
XS Rating Curve= 0 ,0
Exp/Cntr=0.3,0.1

Type RM Length L Ch R = 1 ,32894   ,353,353,353
BEGIN DESCRIPTION:
Mapping XS 985d002d
END DESCRIPTION:
XS GIS Cut Line= 3
      2511381.07     13477647.85      2510552.97     13477548.89
      2509809.11     13477434.45
#Sta/Elev= 30
    4164  218.38  4220.5  217.41  4294.9  214.75    4301  214.37  4310.3  215.36
  4321.2  215.41  4331.3  214.16  4393.5  212.52  4462.2  210.35  4472.2  210.91
  4492.2  209.54  4774.4   202.9  4907.4  202.98  4925.4  202.82  4945.6  201.49
  4965.7  202.49  4975.8  201.25  4994.4   197.5  5014.2  196.95  5014.4  196.45
  5018.2  196.95  5046.5  200.06    5054  202.13  5059.1  202.55  5107.2  202.51
  5329.8  207.14  5592.9  215.51  5648.4  216.55  5673.8  217.92  5750.6  219.67
#Mann= 6 ,-1 , 0
    4164     .07       0  4294.9     .05       0  4393.5    .035       0
  4492.2     .12       0  5014.2     .05       0  5018.2     .12       0
Bank Sta=5014.2,5018.2
XS Rating Curve= 0 ,0
Exp/Cntr=0.3,0.1

Type RM Length L Ch R = 1 ,32541   ,517,517,517
BEGIN DESCRIPTION:
Mapping XS 128f5a27
END DESCRIPTION:
XS GIS Cut Line= 3
      2511257.98     13477293.09      2510619.07     13477272.25
      2510189.22     13477237.59
#Sta/Elev= 30
  4366.2  210.95  4439.2  208.99  4449.2  209.09  4461.8  208.05  4469.2  207.32
  4489.2  208.54  4509.3  207.25    4560  206.22  4699.4  203.59  4729.4  202.66
  4759.4  202.58  4771.1  203.19  4799.4  201.55  4849.4  201.42  4859.4  200.99
  4919.5  201.16  4949.5  199.78  4979.5  200.83  4999.5  195.85    5003  194.05
  5003.2  193.55  5006.7  193.55    5007  194.05    5010  194.05  5019.6  198.04
    5029  199.38    5034  201.66  5099.8  202.13  5270.4  205.08  5436.7  209.36
#Mann= 5 ,-1 , 0
  4366.2     .05       0  4461.8    .035       0    4560     .12       0
    5003     .05       0    5007     .12       0
Bank Sta=5003,5007
XS Rating Curve= 0 ,0
Exp/Cntr=0.3,0.1

Type RM Length L Ch R = 1 ,32024   ,380,380,380
BEGIN DESCRIPTION:
Mapping XS 7b0ed52f
END DESCRIPTION:
XS GIS Cut Line= 3
      2511237.16     13477022.27       2510903.8     13476883.36
      2510349.11     13476827.89
#Sta/Elev= 30
  4648.4  206.75  4672.4  206.07  4684.5  205.22  4702.9  206.24  4707.4     206
  4715.7  204.93  4838.3  202.47  4845.7  201.95  4921.6  200.83  4968.3  199.51
  4992.1   196.9  4997.6  195.47  5004.2  193.02  5004.4  192.52  5007.9  192.52
  5008.2  193.02  5009.5  193.02  5018.4  195.74  5027.4  196.32  5038.4  198.95
  5048.5  199.45  5098.8  199.61  5118.9  200.25  5137.9  200.35  5169.1  201.24
  5244.4  201.94  5344.9  203.76  5380.2  204.93  5440.4  205.67    5567  208.89
#Mann= 6 ,-1 , 0
  4648.4    .035       0  4707.4     .05       0  5004.2     .05       0
  5008.2     .05       0  5027.4      .1       0  5137.9     .12       0
Bank Sta=5004.2,5008.2
XS Rating Curve= 0 ,0
Exp/Cntr=0.3,0.1

Type RM Length L Ch R = 1 ,31644   ,429,429,429
BEGIN DESCRIPTION:
Mapping XS 3b4e27d7
END DESCRIPTION:
XS GIS Cut Line= 3
      2511251.05     13476688.93      2511001.02     13476556.97
       2510542.7     13476508.37
#Sta/Elev= 30
  4690.8  202.19  4697.6  203.18  4706.6  203.76  4712.3  203.65  4720.3  202.63
  4728.6   202.1  4779.2  201.12  4833.1  200.23  4867.2  199.17  4899.1  199.33
  4926.8   198.3  4943.2   198.4  4970.3  197.55  4973.5  196.67  4979.6  195.78
  4989.6  195.35  4999.7  194.26  5007.7   191.2    5008   190.7  5011.5   190.7
  5011.7   191.2  5029.8  195.21  5037.3  197.45  5042.3   198.5  5180.7  201.99
  5232.6  202.67  5251.1  203.61  5381.8  206.73    5412  207.93  5434.4  208.32
#Mann= 4 ,-1 , 0
  4690.8     .05       0  4779.2     .12       0  5007.7     .05       0
  5011.7     .12       0
Bank Sta=5007.7,5011.7
XS Rating Curve= 0 ,0
Exp/Cntr=0.3,0.1

Type RM Length L Ch R = 1 ,31215   ,530,530,530
BEGIN DESCRIPTION:
Mapping XS eddb9235
END DESCRIPTION:
XS GIS Cut Line= 3
       2511598.2     13476293.08      2511119.07     13476181.97
      2510558.25     13476175.05
#Sta/Elev= 30
  4514.2  204.23  4620.8  202.01  4630.4  202.27  4658.3  201.41  4733.1   200.4
  4743.3  200.83  4753.9  200.08  4762.9  200.23  4784.4  198.46  4791.5  199.56
  4815.2  199.77  4834.1  198.04  4878.3  197.67  4979.4  196.59  4989.7  191.16
    4998  189.86  4998.2  189.36  5001.7  189.36    5002  189.86  5005.6  192.56
  5030.1  193.69  5050.1  195.91  5080.1  198.26  5101.4  198.64  5165.6  199.89
  5270.1     203  5390.1  207.68  5470.6  208.85  5530.1  211.59  5566.9  212.66
#Mann= 7 ,-1 , 0
  4514.2     .05       0  4762.9    .035       0  4878.3      .1       0
    4998     .05       0    5002      .1       0  5101.4     .05       0
  5470.6     .12       0
Bank Sta=4998,5002
XS Rating Curve= 0 ,0
Exp/Cntr=0.3,0.1

Type RM Length L Ch R = 1 ,30685   ,607,607,607
BEGIN DESCRIPTION:
Mapping XS f4bae183
END DESCRIPTION:
XS GIS Cut Line= 3
      2511744.11     13475827.82      2511230.18     13475688.92
      2510821.97     13475619.73
#Sta/Elev= 30
  4492.8  199.84  4512.6  200.17  4607.5  198.86  4740.5  198.17  4754.4  197.96
  4771.6  196.66  4781.9  197.61  4794.3  196.67    4813  197.94  4846.3  197.39
  4863.7  196.67  4943.7  195.45  4947.3  195.37    4958  195.33  4968.4  192.57
  4978.1  191.02  4987.1  188.35  4987.4  187.85  4990.9  187.85  4991.1  188.35
  5025.2  192.34  5030.4  194.57  5040.6  195.56  5047.9  195.51  5147.2  197.38
  5192.7  198.14    5198  198.82  5243.4  199.44  5324.6  202.11  5439.2  204.81
#Mann= 9 ,-1 , 0
  4492.8     .07       0  4607.5     .05       0  4846.3      .1       0
  4943.7     .12       0  4947.3      .1       0  4987.1     .05       0
  4991.1      .1       0  5047.9     .12       0  5147.2     .05       0
Bank Sta=4987.1,4991.1
XS Rating Curve= 0 ,0
Exp/Cntr=0.3,0.1

Type RM Length L Ch R = 1 ,30078   ,432,432,432
BEGIN DESCRIPTION:
KILGORE CREEK 59.0
END DESCRIPTION:
XS GIS Cut Line= 3
        2511925.       13475325.        2511375.       13475125.
      2510925.01       13475225.
#Sta/Elev= 30
  4409.4  201.46  4424.7  202.21  4430.7  201.27  4558.4  198.35  4653.5  197.43
  4689.4  196.39  4707.3  196.81  4714.7  196.08  4739.3  195.94  4745.2  196.49
  4760.5  195.68  4792.5  195.21  4856.3  194.96  4947.1  193.65  4962.7  193.73
  4984.7  190.17  4997.2  190.18  5004.9  187.45  5016.9  186.66  5017.2  186.16
  5020.8  186.16    5021  186.66  5025.4  188.88  5035.6  192.71  5045.9  193.71
  5150.8  194.83  5168.8  195.69  5189.3  195.15  5240.5  195.98  5455.6  201.66
#Mann= 5 ,-1 , 0
  4409.4     .05       0  4947.1     .07       0  5016.9     .05       0
    5021     .07       0  5150.8     .05       0
Bank Sta=5016.9,5021
XS Rating Curve= 0 ,0
Exp/Cntr=0.3,0.1

Type RM Length L Ch R = 1 ,29646   ,460,460,460
BEGIN DESCRIPTION:
KILGORE CREEK 58.0
END DESCRIPTION:
XS GIS Cut Line= 3
        2511925.       13474825.        2511425.       13474775.
        2511025.       13474875.
#Sta/Elev= 30
  4491.9  198.94  4612.5  196.58  4632.6  196.69  4645.2  195.81  4693.9  195.52
  4702.9  195.82    4713  195.09  4792.4  193.86  4813.5  194.03    4914  191.75
  4954.2  191.81  4974.3  188.85    4997  190.19  5012.4  185.73  5017.6  187.69
  5023.2   184.2  5023.5   183.7  5027.1   183.7  5027.4   184.2  5035.6  184.52
  5053.7  191.24  5058.8  189.89  5066.5  191.81    5100   192.6  5107.8  193.46
  5141.3   193.4  5193.3   194.8    5265  196.48    5283  198.22  5406.7  198.59
#Mann= 6 ,-1 , 0
  4491.9     .05       0  4693.9     .07       0  4792.4     .12       0
  5023.2     .05       0  5027.4     .12       0  5193.3    .094       0
Bank Sta=5023.2,5027.4
XS Rating Curve= 0 ,0
Exp/Cntr=0.3,0.1

Type RM Length L Ch R = 1 ,29186   ,362,362,362
BEGIN DESCRIPTION:
KILGORE CREEK 57.0
END DESCRIPTION:
XS GIS Cut Line= 3
      2511924.98       13474425.        2511575.       13474375.
      2510975.03       13474375.
#Sta/Elev= 30
  4646.5  198.23  4655.5  197.93    4697  197.32  4707.1  197.69  4737.4  196.63
  4767.7  194.44  4818.2  193.52  4860.2  192.04    4899   191.7  4939.4  192.11
  4949.5   191.7  4959.6   190.2  4969.7   186.8  4977.7  183.13    4978  182.63
  4981.7  182.63    4982  183.13  4989.9  184.63  4997.5  188.71  5002.5  188.71
    5010  189.82    5030  190.86    5110  190.48    5190  191.34    5210  191.96
  5245.2  192.04  5428.7  195.42    5550  197.64    5570  198.94    5600  199.49
#Mann= 7 ,-1 , 0
  4646.5     .05       0  4655.5     .07       0  4860.2     .12       0
  4977.7     .05       0    4982     .12       0  5245.2     .05       0
  5428.7     .12       0
Bank Sta=4977.7,4982
XS Rating Curve= 0 ,0
Exp/Cntr=0.3,0.1

Type RM Length L Ch R = 1 ,28824   ,138,138,138
BEGIN DESCRIPTION:
Mapping XS 8ecb7ea6
END DESCRIPTION:
XS GIS Cut Line= 3
      2512084.11     13474232.64      2511476.49     13474045.15
      2510820.24     13474114.59
#Sta/Elev= 30
  4362.2   200.3  4384.1  199.68  4424.1  198.61  4455.5  198.69    4472  197.44
  4497.3  197.64  4591.5  194.67  4645.8  194.13  4775.2  191.24  4853.1  188.69
    4895  189.81  4905.5  189.53  4912.2  188.01  4936.9   187.9  4977.6  185.57
  4989.2  185.89  4994.1  182.95  4994.4  182.45  4998.2  182.45  4998.4  182.95
  5004.7  182.99  5009.6  183.04  5019.7  186.27  5044.5  190.29  5180.6  191.22
  5387.8  195.03  5420.6  196.47  5523.4  198.87  5633.1  202.21    5658  202.24
#Mann= 7 ,-1 , 0
  4362.2     .12       0  4384.1     .07       0  4775.2     .12       0
  4994.1     .05       0  4998.4     .12       0  5004.7     .05       0
  5387.8     .12       0
Bank Sta=4994.1,4998.4
XS Rating Curve= 0 ,0
Exp/Cntr=0.3,0.1

Type RM Length L Ch R = 1 ,28686   ,176,176,176
BEGIN DESCRIPTION:
Mapping XS 026ccb17
END DESCRIPTION:
XS GIS Cut Line= 3
      2512226.78     13474173.39      2511495.48     13473917.33
      2510818.08     13474012.55
#Sta/Elev= 30
  4293.4  203.49  4401.2  201.63  4426.2  200.63  4528.4  199.13  4560.2  199.48
  4570.7   198.4  4613.1  196.98  4687.4  195.32  4750.9  193.12  4844.6  190.85
  4849.9  191.37  4860.9  188.99  4888.6  185.56  4899.2  185.49  4920.4  186.89
    4943  185.96  4962.8  186.08    4974  184.19  4994.5  184.46  5013.6  182.04
  5013.9  181.54  5017.7  181.54  5017.9  182.04  5025.5  182.52  5030.8  184.99
    5037  189.51  5054.5  189.41  5260.6  190.91  5442.1  193.96  5752.3  202.08
#Mann= 7 ,-1 , 0
  4293.4     .12       0  4687.4     .07       0  4860.9     .12       0
  5013.6     .05       0  5017.9     .12       0  5054.5     .05       0
  5442.1     .12       0
Bank Sta=5013.6,5017.9
XS Rating Curve= 0 ,0
Exp/Cntr=0.3,0.1

Type RM Length L Ch R = 1 ,28510   ,280,280,280
BEGIN DESCRIPTION:
Mapping XS 375439d7
END DESCRIPTION:
XS GIS Cut Line= 3
      2512254.24     13473937.51      2511667.46     13473829.87
      2510809.92      13473961.8
#Sta/Elev= 30
  4409.2  203.85  4469.4  203.37  4540.6  200.14  4563.8  200.38  4571.1  199.69
  4713.4  197.18  4743.9  195.73  4845.6  193.78  4876.1  191.94  4957.4  189.97
  4987.9  187.56  4998.1  185.38  5004.1  180.79  5007.8  180.53  5008.1  180.03
  5012.2  180.53  5018.4  183.08  5028.5  185.33  5038.6   186.4  5068.1  185.62
  5073.2  187.04  5089.2  185.83  5109.4  186.62  5129.7  188.76  5144.4  188.75
  5476.4  192.25  5564.7  193.64  5645.7  196.52  5862.4   200.9  5873.4  201.93
#Mann= 5 ,-1 , 0
  4409.2     .12       0  5007.8     .05       0  5012.2     .12       0
  5144.4     .05       0  5476.4     .12       0
Bank Sta=5007.8,5012.2
XS Rating Curve= 0 ,0
Exp/Cntr=0.3,0.1

Type RM Length L Ch R = 1 ,28230   ,318,318,318
BEGIN DESCRIPTION:
Mapping XS 94c0d51f
END DESCRIPTION:
XS GIS Cut Line= 3
      2512268.12     13473645.84      2511632.74     13473593.76
      2510640.47     13473840.09
#Sta/Elev= 30
  4354.3  201.34  4424.2  200.67  4437.7  199.97    4463  199.69  4568.1  197.31
  4658.4  195.87  4688.5  194.41  4788.4  192.48  4798.9  191.51    4839  190.18
  4869.1  190.29  4889.2  189.45  4919.9  189.16  4949.4  187.11  4969.5  180.63
  4977.3  180.34  4977.6  179.84  4981.4  179.84  4981.7  180.34  4988.2  183.42
  4991.8  183.42  4999.8  186.04  5016.5  187.41  5057.8  188.67  5140.6  187.69
  5236.8   188.1  5600.7  193.84  5779.6  198.17  5983.6  204.21  6014.2  204.41
#Mann= 6 ,-1 , 0
  4354.3     .07       0    4463     .12       0  4977.3     .05       0
  4981.7     .12       0  5779.6     .07       0  5983.6     .05       0
Bank Sta=4977.3,4981.7
XS Rating Curve= 0 ,0
Exp/Cntr=0.3,0.1

Type RM Length L Ch R = 1 ,27912   ,1130,1130,1130
BEGIN DESCRIPTION:
Mapping XS 0aa26b89
END DESCRIPTION:
XS GIS Cut Line= 3
      2512250.87     13473335.35       2511573.8     13473324.94
      2510699.43      13473507.1
#Sta/Elev= 30
  4328.6  194.05  4454.5  193.14  4484.5   192.4  4514.5  192.55  4742.3  189.85
  4914.5  187.72  4964.5  186.22  4974.5  185.19  4984.5  183.44  4994.5  181.03
  5000.4  178.37  5000.7  177.87  5004.5  177.87  5004.8  178.37  5014.7  181.06
    5025  181.31  5030.3  186.31  5045.4  187.21  5116.9  186.77  5165.6  184.54
  5180.5  184.21  5188.4   183.3  5249.7  187.32  5325.1   188.1  5484.6  190.92
  5545.9  192.76  5556.1  193.54  5576.5  193.44  5780.8  198.75  5898.9  200.69
#Mann= 6 ,-1 , 0
  4328.6    .035       0  4742.3     .12       0  5000.4     .05       0
  5004.8     .12       0  5165.6    .035       0  5325.1     .12       0
Bank Sta=5000.4,5004.8
XS Rating Curve= 0 ,0
Exp/Cntr=0.3,0.1

Type RM Length L Ch R = 1 ,26782   ,207,207,207
BEGIN DESCRIPTION:
Mapping XS e208d35f
END DESCRIPTION:
XS GIS Cut Line= 4
      2512355.07     13472653.06       2511256.1      13472741.6
       2510948.8     13472887.44      2510422.78     13473444.71
#Sta/Elev= 30
  3915.5  199.76  4089.3  196.55  4131.2  195.52  4291.4  192.92  4818.5   185.7
  4868.6  183.61  4873.6  182.43  4888.7  184.38  4908.8  181.73  4938.9  181.97
    4969  180.23    4979  180.67  4993.6   175.3    4994   174.8  4998.5   175.3
  5009.1  178.41  5016.1  179.32  5030.3  178.76  5058.9  184.53    5141  186.48
  5195.9  186.67  5254.1  187.69    5310   188.4  5493.4  191.79  5521.7  192.51
    5529   193.5    5550  193.28  5599.8  194.83  5974.4  200.39  6124.5  201.37
#Mann= 10 ,-1 , 0
  3915.5     .07       0  4089.3    .035       0  4131.2     .07       0
  4291.4     .12       0  4993.6     .05       0  4998.5     .12       0
  5058.9     .07       0  5195.9     .12       0  5254.1     .07       0
    5310     .12       0
Bank Sta=4993.6,4998.5
XS Rating Curve= 0 ,0
Exp/Cntr=0.3,0.1

Type RM Length L Ch R = 1 ,26575   ,715,715,715
BEGIN DESCRIPTION:
Mapping XS fdc6c7ca
END DESCRIPTION:
XS GIS Cut Line= 4
      2512079.88     13472518.54      2511353.35     13472505.52
      2511176.27     13472565.42      2510596.98     13473051.19
#Sta/Elev= 30
  4137.6  196.01  4428.9  189.95  4622.6  185.98  4722.6  185.68  4832.6  183.65
  4904.4   183.2  4915.3  182.58  4925.8  180.67  4935.9  179.94  4957.5   179.4
  4972.6  179.87  4989.2   178.1  4996.3  174.04  4996.7  173.54  5001.2  174.04
  5010.3  175.19  5020.9  177.69  5030.2  184.78  5071.2  185.29  5112.8   185.5
  5144.2  186.36  5157.7   185.9    5326  187.19  5417.1  187.91  5474.5  188.73
  5548.5  190.05  5622.9  191.46  5665.3  191.89  5796.7  193.38  5807.2  194.05
#Mann= 12 ,-1 , 0
  4137.6     .07       0  4428.9     .12       0  4996.3     .05       0
  5001.2     .12       0  5071.2     .07       0  5112.8     .12       0
    5326     .07       0  5417.1      .1       0  5474.5     .07       0
  5548.5      .1       0  5622.9     .07       0  5665.3     .12       0
Bank Sta=4996.3,5001.2
XS Rating Curve= 0 ,0
Exp/Cntr=0.3,0.1

Type RM Length L Ch R = 1 ,25860   ,442,442,442
BEGIN DESCRIPTION:
Mapping XS a4e73e07
END DESCRIPTION:
XS GIS Cut Line= 4
      2512615.48     13472377.02      2511681.47     13472083.65
      2510960.12     13472039.38      2510004.42     13472195.62
#Sta/Elev= 30
  3908.9  206.12  4108.6  204.61  4198.5  201.79  4378.8  198.66  4661.9   191.3
    4764   188.8  4866.1  186.97  4954.5  185.03  4984.6  179.22  5004.6     177
  5014.6  173.11  5022.2  172.75  5022.5  172.25  5027.1  172.75  5034.6  176.69
  5044.7  177.24  5063.6  181.27  5084.7  182.08  5124.8  180.28    5235  183.28
  5346.4     183  5357.4  183.04  5399.4  182.71  5475.5  181.57  5505.5  178.51
  5525.6  174.59  5545.6   184.4  5696.9  185.48  6039.5  190.76    6579  199.31
#Mann= 11 ,-1 , 0
  3908.9     .05       0  4378.8     .12       0  4661.9    .035       0
    4764     .12       0  4866.1     .07       0  5022.2     .05       0
  5063.6      .1       0  5346.4    .035       0  5357.4      .1       0
  5399.4    .035       0  6039.5     .07       0
#XS Ineff= 2 , 0
       0                  5265.1       0     190
Permanent Ineff=
       F       F
Bank Sta=5022.2,5027.1
XS Rating Curve= 0 ,0
Exp/Cntr=0.3,0.1

Type RM Length L Ch R = 1 ,25418   ,851,851,851
BEGIN DESCRIPTION:
Mapping XS fe7641b2
END DESCRIPTION:
XS GIS Cut Line= 3
      2512516.51     13471830.14      2511412.35     13471752.02
      2509974.81     13471580.14
#Sta/Elev= 30
  3905.5   198.6  4027.3  198.06  4077.4  196.52  4127.6  197.08  4221.1  195.04
  4516.2  188.14  4624.4  185.29  4712.9  183.36  4849.4  181.49  4879.4  179.44
    4932  179.04  4959.6  174.15  5004.8  170.78  5005.3  170.28  5012.4  170.78
  5027.1  171.95  5032.2  170.93    5050  174.04  5060.1  173.39  5070.2  171.06
  5090.3  173.95  5109.6  182.61  5114.6  183.17  5205.2  182.72  5284.4  182.22
  5311.9  184.21  5339.4  183.58  5493.2  184.64  5755.5   189.4  6460.2  199.05
#Mann= 11 ,-1 , 0
  3905.5     .05       0  4221.1     .07       0  4516.2    .035       0
  4624.4     .12       0  4712.9     .07       0    4932    .063       0
  5004.8     .05       0  5012.4    .063       0  5205.2     .07       0
  5339.4     .05       0  5755.5     .07       0
Bank Sta=5004.8,5012.4
XS Rating Curve= 0 ,0
Exp/Cntr=0.3,0.1

Type RM Length L Ch R = 1 ,24567   ,596,596,596
BEGIN DESCRIPTION:
Mapping XS dcead758
END DESCRIPTION:
XS GIS Cut Line= 3
      2512549.52     13471203.41      2511757.83     13471147.85
      2510259.13     13471369.88
#Sta/Elev= 30
  4249.5  197.52  4285.5  196.92  4374.3  193.34  4424.5  198.77  4464.6  193.68
    4635  189.93  4675.1  190.71  4685.1   188.4  4725.9  188.39  4925.7  182.92
  4945.7  179.37  4965.8  168.83  4971.9  167.95  4972.4  167.45  4979.7  167.95
  4985.8  167.95  5011.7  178.38  5018.3  177.37  5059.5   180.2  5217.9  180.18
  5264.7  176.39  5272.4  175.96  5277.4  176.13  5308.8  179.37  5453.1  181.61
    5557  182.07  5795.1  184.01  6148.2  188.31  6318.1  190.64  6558.2  194.31
#Mann= 14 ,-1 , 0
  4249.5     .12       0  4285.5     .07       0  4725.9    .035       0
  4971.9     .05       0  4979.7    .035       0  5018.3     .07       0
  5264.7     .05       0  5272.4     .07       0  5277.4     .05       0
  5453.1     .07       0    5557     .05       0  5795.1     .07       0
  6148.2    .035       0  6318.1     .07       0
Bank Sta=4971.9,4979.7
XS Rating Curve= 0 ,0
Exp/Cntr=0.3,0.1

Type RM Length L Ch R = 1 ,23971   ,938,938,938
BEGIN DESCRIPTION:
Mapping XS 734f616a
END DESCRIPTION:
XS GIS Cut Line= 3
      2512653.71     13470606.19        2511612.     13470613.13
      2510279.36     13470765.83
#Sta/Elev= 30
  3958.5  195.39  4047.2  193.09  4099.2  192.49  4277.2  188.58  4531.4  184.87
    4770  179.36  4867.2  178.82  4947.2  177.03  4957.2  176.44  4966.7  173.51
  5013.4  167.28  5013.9  166.78  5020.8  166.78  5021.3  167.28  5027.4   167.7
  5037.5  171.89  5047.5  173.15  5067.7  172.28  5077.7  173.06  5093.4  175.64
  5107.9  177.93    5118  178.73  5138.1  179.26  5150.8  178.15  5208.6  180.76
  5413.5  181.85  5822.6  183.87  5902.3  185.25  6173.4  188.55  6341.6  192.81
#Mann= 10 ,-1 , 0
  3958.5     .07       0  4099.2     .05       0    4770     .07       0
  4966.7      .1       0  5013.4     .05       0  5021.3      .1       0
  5093.4     .07       0  5413.5     .05       0  5902.3     .07       0
  6173.4     .05       0
Bank Sta=5013.4,5021.3
XS Rating Curve= 0 ,0
Exp/Cntr=0.3,0.1

Type RM Length L Ch R = 1 ,23033   ,717,717,717
BEGIN DESCRIPTION:
Mapping XS 2c990f24
END DESCRIPTION:
XS GIS Cut Line= 3
      2512799.53     13469932.57      2511709.22     13469981.19
      2510264.78     13470182.57
#Sta/Elev= 30
  3884.1  203.01  3928.7  201.62  4008.7   200.7  4158.9  196.14  4178.9  196.24
    4309  192.58  4409.1  190.89  4445.4  189.03  4609.3  185.29  4869.1  176.38
  4879.6  176.07  4919.7  170.96  4939.7  169.59  4946.8  166.06  4951.8  165.42
  4970.9  164.88  4971.4  164.38  4979.3  164.88    5010  174.26  5020.1  175.83
  5071.2  177.06  5222.1  177.28  5493.2  179.37  5670.9  180.34  5706.7  181.41
  5726.9  180.65  5938.3  183.29  6060.1  185.47  6116.5  185.63  6433.9  192.23
#Mann= 10 ,-1 , 0
  3884.1     .12       0  4445.4     .07       0  4869.1    .035       0
  4970.9     .05       0  4979.3    .035       0  5071.2     .07       0
  5493.2    .035       0  5670.9     .05       0  5938.3     .07       0
  6116.5     .05       0
Bank Sta=4970.9,4979.3
XS Rating Curve= 0 ,0
Exp/Cntr=0.3,0.1

Type RM Length L Ch R = 1 ,22316   ,774,774,774
BEGIN DESCRIPTION:
Mapping XS 676e2aa5
END DESCRIPTION:
XS GIS Cut Line= 3
      2512862.02      13469467.3       2511674.5     13469335.35
       2510328.6     13469598.98
#Sta/Elev= 30
  3805.6  203.88  3908.8  202.51    4316     192  4401.8  189.89  4687.9  183.27
  4929.5  177.57  4949.6  173.69  4956.5  169.02  4961.5  170.52  4969.7  166.88
  4985.6  163.39  4986.1  162.89  4994.1  163.39  5002.7  163.74  5010.1  168.02
  5030.5  171.28  5091.6  174.01  5142.6  174.83  5193.5  172.46  5254.7  175.39
  5377.4  176.32    5396  176.44  5647.9  177.76  5723.4  176.72  5733.6  178.48
  5752.5  177.39  5899.6  181.02  6000.3  183.45  6272.6  190.39  6371.9  193.23
#Mann= 13 ,-1 , 0
  3805.6     .05       0  3908.8     .12       0    4316     .07       0
  4401.8     .05       0  4687.9     .07       0  4985.6     .05       0
  4994.1     .07       0  5377.4    .063       0    5396    .094       0
  5752.5     .07       0  5899.6    .094       0  6000.3     .05       0
  6272.6     .07       0
Bank Sta=4985.6,4994.1
XS Rating Curve= 0 ,0
Exp/Cntr=0.3,0.1

Type RM Length L Ch R = 1 ,21542   ,514,514,514
BEGIN DESCRIPTION:
Mapping XS abbfea54
END DESCRIPTION:
XS GIS Cut Line= 4
      2512806.47     13469029.81      2511556.44     13468675.63
      2511243.94     13468689.52      2510238.49     13469001.56
#Sta/Elev= 30
  3480.1  197.23  3516.3  196.56  3937.1   188.8  4425.9  180.24  4694.1  175.94
  4840.8   175.1  4860.9  168.54  4870.9  167.77  4876.8  170.78  4890.9  167.57
  4900.9  169.69  4930.9  169.69  4950.9  167.18    4961  163.55  4986.5  161.99
    4987  161.49  4995.4  161.99    5011  165.46  5071.1  167.37  5089.1  172.34
  5092.1  172.34    5095  169.93  5101.5  171.86  5358.1  176.89  5475.5  180.44
  5747.9  186.41    6006   193.6  6043.9  195.76  6071.1  195.24  6144.9   197.5
#Mann= 10 ,-1 , 0
  3480.1     .05       0  3516.3     .12       0  3937.1     .05       0
  4425.9     .07       0  4694.1     .12       0  4986.5     .05       0
  4995.4     .12       0  5358.1     .05       0  5475.5     .07       0
  5747.9     .05       0
Bank Sta=4986.5,4995.4
XS Rating Curve= 0 ,0
Exp/Cntr=0.3,0.1

Type RM Length L Ch R = 1 ,21028   ,514,514,514
BEGIN DESCRIPTION:
Mapping XS 52445414
END DESCRIPTION:
XS GIS Cut Line= 4
      2512827.29     13468758.97      2511563.39     13468196.46
      2511084.22      13468217.3      2510258.94      13468494.7
#Sta/Elev= 30
  3377.7  196.04  3429.9  194.59  3536.1  191.91  3656.8  188.56  3748.6  186.39
  3915.8  182.82  4173.6  179.64  4174.8  179.64  4279.9  179.68  4386.1  178.33
  4433.8   177.7  4683.8  172.99  4717.8   172.4  4929.7  172.34  4979.7  166.91
  4989.7  164.09  4995.3  160.67  4995.8  160.17  5004.2  160.67  5012.4  162.19
  5019.8  165.75  5029.8  166.51  5049.8  165.39  5100.9  166.79  5149.9  164.53
  5209.9  168.54  5237.9  174.32  5622.5  187.24  5756.9  190.57  6111.4   195.1
#Mann= 18 ,-1 , 0
  3377.7     .05       0  3429.9     .07       0  3536.1     .12       0
  3656.8     .07       0  3748.6     .12       0  3915.8     .07       0
  4173.6    .035       0  4174.8     .07       0  4279.9    .035       0
  4386.1     .07       0  4433.8     .12       0  4683.8     .07       0
  4717.8     .12       0  4995.3     .05       0  5004.2     .12       0
  5012.4     .07       0  5100.9     .12       0  5622.5     .05       0
Bank Sta=4995.3,5004.2
XS Rating Curve= 0 ,0
Exp/Cntr=0.3,0.1

Type RM Length L Ch R = 1 ,20514   ,950,950,950
BEGIN DESCRIPTION:
Mapping XS 20cfc608
END DESCRIPTION:
XS GIS Cut Line= 3
      2512834.23     13468439.52      2511521.72     13467765.91
       2510535.6     13467196.46
#Sta/Elev= 30
  3497.1   194.3    3542  193.41  3543.2  193.43  3619.9  192.78  3664.8  188.73
  3709.6  192.36    3766  188.73  4145.5  180.74  4397.5  176.57  4642.7  166.42
  4658.2  168.99    4697  166.95  4702.6  168.99  4719.1  166.09  4763.5  167.13
  4769.1  165.22  4777.6   169.6  4807.9  166.64  4830.1  170.11  4877.4  170.17
  4955.3  165.69  4979.3  165.23  4995.9  159.28  4996.4  158.78  5005.7  159.28
  5028.1  168.03  5075.5  171.88  5644.1  186.41  6080.7  190.27  6111.1  190.69
#Mann= 10 ,-1 , 0
  3497.1     .05       0    3542     .07       0  3543.2     .05       0
  4145.5     .12       0  4877.4     .07       0  4955.3      .1       0
  4995.9     .05       0  5005.7      .1       0  5075.5     .12       0
  6080.7     .07       0
Bank Sta=4995.9,5005.7
XS Rating Curve= 0 ,0
Exp/Cntr=0.3,0.1

Type RM Length L Ch R = 1 ,19564   ,720,720,720
BEGIN DESCRIPTION:
Mapping XS eff3c52d
END DESCRIPTION:
XS GIS Cut Line= 3
      2513021.73      13467717.3      2512264.78     13467307.58
       2511070.3     13467085.35
#Sta/Elev= 30
  4150.1  191.02  4349.9  186.23  4385.2  183.86  4421.3  184.38  4499.1   182.6
  4609.2  180.59  4967.3  172.69  4976.5  171.04  4983.4  163.83  4989.1  162.18
  5000.3     157  5000.8   156.5  5010.4     157  5010.8  158.06  5013.3  158.06
  5020.8  161.69  5030.9  162.98  5041.1  162.19  5061.5  164.38    5102  165.95
    5153  166.13    5174  167.92  5270.5  170.06  5427.6  168.26  5491.7   169.2
  5590.4  172.18  5773.5  180.71  5813.4  180.87  5854.8  182.72  6225.8  190.36
#Mann= 6 ,-1 , 0
  4150.1    .035       0  4499.1     .07       0  4609.2     .12       0
  5000.3     .05       0  5010.4     .12       0    5174     .05       0
Bank Sta=5000.3,5010.4
XS Rating Curve= 0 ,0
Exp/Cntr=0.3,0.1

Type RM Length L Ch R = 1 ,18844   ,719,719,719
BEGIN DESCRIPTION:
Mapping XS 14e413d3
END DESCRIPTION:
XS GIS Cut Line= 3
      2513348.11     13466821.46      2512243.94     13466640.91
      2511168.78     13466682.53
#Sta/Elev= 30
  3862.2   186.7  4128.8  178.74  4280.8  176.56  4382.1  174.13  4617.6   170.6
  4796.6  170.59  4863.1  169.25    4909  167.91  4949.6  163.96  4969.8  160.59
    4978  157.85  4994.9  154.81  4995.4  154.31  5005.1  154.81    5020  159.91
    5030  160.81    5050   165.4  5080.1  166.26  5090.1  164.68  5100.1  161.21
  5121.7  162.77  5170.1  166.77    5475  174.22  5690.5  183.42  5760.6  184.39
  5850.6   186.7  5890.7  188.57  5970.7  189.74  5980.7  190.66    6057  191.68
#Mann= 4 ,-1 , 0
  3862.2     .12       0  4994.9     .05       0  5005.1     .12       0
  5121.7     .05       0
Bank Sta=4994.9,5005.1
XS Rating Curve= 0 ,0
Exp/Cntr=0.3,0.1

Type RM Length L Ch R = 1 ,18125   ,457,457,457
BEGIN DESCRIPTION:
Mapping XS 94ffd553
END DESCRIPTION:
XS GIS Cut Line= 3
      2513445.37      13466217.3      2512348.11     13465981.19
       2511132.8     13466022.85
#Sta/Elev= 30
  3854.4  186.77  4354.9  173.87  4399.6   172.5  4673.1  166.19  4840.8  164.36
  4928.8  164.87  4949.3  163.67  4959.5  161.53  4975.8  153.37  4984.5  153.21
    4985  152.71  4995.2  153.21  4999.9  153.54  5019.9  158.61  5039.9  160.57
  5059.9  157.92    5090  160.71    5120  164.39    5140  168.45    5150   171.5
    5160  172.28    5200  164.04  5229.5  160.45  5269.8  164.33  5290.1  168.55
  5300.1  169.12  5650.3  175.22  5980.4  185.23  6047.1  186.86  6192.8  190.24
#Mann= 8 ,-1 , 0
  3854.4     .12       0  4354.9     .05       0  4399.6     .12       0
  4984.5     .05       0  4995.2     .12       0  5269.8     .05       0
  5980.4     .12       0  6047.1     .05       0
Bank Sta=4984.5,4995.2
XS Rating Curve= 0 ,0
Exp/Cntr=0.3,0.1

Type RM Length L Ch R = 1 ,17668   ,520,520,520
BEGIN DESCRIPTION:
Mapping XS fffce112
END DESCRIPTION:
XS GIS Cut Line= 3
      2513334.21     13465821.46      2512396.72     13465543.69
      2511349.01     13465418.79
#Sta/Elev= 30
  4000.3  182.59  4082.9  179.29  4463.9  168.55  4678.4  162.84  4783.4  164.26
  4849.9     164  4888.3  162.55  4921.6  163.54  4954.8  159.65  4969.4     159
  4976.4   156.7  4981.5   156.7  4994.6  152.56  4995.1  152.06  5005.4  152.56
  5030.2  157.33  5070.4  159.36  5089.6  162.85  5094.7  160.58  5110.7  164.37
  5291.2  169.89  5489.9  175.97  5644.5  179.59  5682.4     181    5715  183.87
    5765  183.35    5770   184.9  5825.8   183.4    5935  185.86  6033.2   186.7
#Mann= 7 ,-1 , 0
  4000.3     .05       0  4463.9     .12       0  4994.6     .05       0
  5005.4     .12       0  5291.2    .035       0  5489.9      .1       0
    5765     .12       0
Bank Sta=4994.6,5005.4
XS Rating Curve= 0 ,0
Exp/Cntr=0.3,0.1

Type RM Length L Ch R = 1 ,17148   ,218,218,218
BEGIN DESCRIPTION:
Mapping XS bd566afd
END DESCRIPTION:
XS GIS Cut Line= 3
      2513368.95     13465710.36       2512674.5     13465189.52
      2511521.75     13464536.76
#Sta/Elev= 30
  4121.8  183.04  4356.9  177.29  4635.9  168.28  4864.2  161.87  4927.7  161.56
  4977.5  155.82  4979.4  155.61    4986  154.84  4989.5  151.64  5002.4  151.26
  5002.9  150.76  5013.3  151.26  5013.6  153.39  5023.8   154.5  5029.5  156.34
  5051.1  158.48  5094.4  160.14  5110.3   158.7  5131.9  159.21  5147.8  161.55
  5169.5  162.97  5198.9  163.02  5336.6  164.64  5417.7  165.64  5595.2  172.98
  5805.8  179.88  6092.5  185.08  6138.5  185.13  6218.9  187.28  6314.6  187.44
#Mann= 8 ,-1 , 0
  4121.8     .05       0  4635.9     .12       0  4977.5    .035       0
  4979.4     .12       0  5002.4     .05       0  5013.3     .12       0
  5198.9    .035       0  5336.6     .05       0
Bank Sta=5002.4,5013.3
XS Rating Curve= 0 ,0
Exp/Cntr=0.3,0.1

Type RM Length L Ch R = 1 ,16930   ,263,263,263
BEGIN DESCRIPTION:
Mapping XS c1df8b45
END DESCRIPTION:
XS GIS Cut Line= 3
      2513792.95     13465642.96      2512827.28     13465036.74
      2511601.57      13464279.2
#Sta/Elev= 30
  3812.9  192.81  3852.7  191.57    3861   191.3  4191.4   182.9  4295.9  180.51
  4629.7  172.09  4708.1  170.09  4877.8   160.1  4896.7  157.37  4911.9  157.44
  4927.2  160.68  4942.5  159.57  4951.5  155.15  4957.4  155.15  4969.7  151.19
  4979.6  149.62  4980.1  149.12  4990.5  149.62  5018.9  158.03  5027.6  160.35
    5043   161.5  5079.6  162.16  5369.2  162.22  5537.1   165.4  5943.2  179.02
    6002  179.64  6015.9  178.81  6073.8  181.22  6162.5  181.97    6394  181.29
#Mann= 10 ,-1 , 0
  3812.9    .035       0  3852.7     .12       0    3861    .035       0
  4191.4     .12       0  4295.9    .035       0  4629.7     .05       0
  4877.8    .063       0  4979.6     .05       0  4990.5    .063       0
  5018.9    .035       0
Bank Sta=4979.6,4990.5
XS Rating Curve= 0 ,0
Exp/Cntr=0.3,0.1

Type RM Length L Ch R = 1 ,16667   ,400,400,400
BEGIN DESCRIPTION:
Mapping XS f1899f18
END DESCRIPTION:
XS GIS Cut Line= 3
      2513654.47     13465311.66        2512960.     13464834.21
      2511775.08     13464287.33
#Sta/Elev= 30
  4161.5  187.58  4201.5  187.55  4216.4  186.29    4283  184.89    4386  182.54
    4503  178.73  4759.4  168.73  4864.6  164.53  4949.7  159.42  4963.3  157.08
  4972.1  157.25  4986.1  150.49  4993.7  149.19  4994.2  148.69  5004.7  149.19
  5009.3  149.45  5015.7   151.6  5031.8  155.39  5060.7  159.73  5106.6   162.1
  5203.9  160.54  5241.1  161.89  5329.6  160.46  5495.7  161.52  5707.7  166.56
  5919.8  174.89    6017  176.38  6062.9  178.47  6154.7  180.24  6309.3  179.97
#Mann= 8 ,-1 , 0
  4161.5     .12       0    4283     .05       0    4386     .07       0
    4503     .05       0  4759.4     .12       0  4993.7     .05       0
  5004.7     .12       0  5015.7     .05       0
Bank Sta=4993.7,5004.7
XS Rating Curve= 0 ,0
Exp/Cntr=0.3,0.1

Type RM Length L Ch R = 1 ,16267   ,508,508,508
BEGIN DESCRIPTION:
Mapping XS 46b7b315
END DESCRIPTION:
XS GIS Cut Line= 3
      2514037.82     13465143.14      2513246.11       13464532.
      2511940.51     13464094.49
#Sta/Elev= 30
  3872.3     196  3969.5  192.39  4203.4  185.44  4218.6  184.98  4330.5  183.01
  4445.4  179.64    4504  178.02  4664.2  173.98  4929.4  164.03  4973.5  162.32
  4979.1  156.85  4989.6  149.84  5005.2  148.03  5005.7  147.53  5016.2  148.03
  5021.3  151.74  5031.3   153.8  5084.5  156.25  5131.3  154.77  5157.5     159
  5192.7  160.17  5257.5  157.34  5315.3  157.21  5441.4   160.2  5583.3  161.56
  5749.4  165.36  5892.2  169.66  5951.2  172.54  6054.8   175.5  6249.4  175.91
#Mann= 16 ,-1 , 0
  3872.3     .05       0  3969.5    .035       0  4203.4     .05       0
  4218.6     .07       0  4330.5     .12       0  4445.4     .07       0
    4504     .12       0  4929.4     .05       0  5005.2     .05       0
  5016.2     .05       0  5192.7     .07       0  5441.4     .05       0
  5583.3     .12       0  5749.4     .05       0  5892.2    .035       0
  5951.2     .05       0
Bank Sta=5005.2,5016.2
XS Rating Curve= 0 ,0
Exp/Cntr=0.3,0.1

Type RM Length L Ch R = 1 ,15759   ,335,335,335
BEGIN DESCRIPTION:
Mapping XS c704e2c9
END DESCRIPTION:
XS GIS Cut Line= 3
      2514110.13     13464612.84      2512964.34      13464035.6
      2512091.98     13463631.97
#Sta/Elev= 30
  3729.4  190.77  3767.8  189.67  3984.8  184.18  4093.4   180.9    4117  180.22
  4229.1   176.8    4239  175.06  4310.4  174.88  4527.4  167.81  4581.5  166.22
  4630.9  162.08  4714.3  158.86  4889.3  158.26    4982  152.82  4993.2  146.98
  4993.7  146.48  5004.3  146.98  5014.8   147.5    5035  157.34  5044.4  160.41
  5055.7  161.01  5176.1  162.57    5336  162.83  5606.7  166.53  5645.1  163.66
  5690.9  165.42  5705.8  167.79  5736.8   166.2    5811     169  5973.6   171.2
#Mann= 13 ,-1 , 0
  3729.4     .07       0  3767.8    .035       0  3984.8     .07       0
  4093.4     .12       0    4117     .07       0  4310.4     .12       0
  4527.4    .035       0  4581.5     .12       0  4889.3     .05       0
  4993.2     .05       0  5004.3     .05       0    5035     .07       0
  5176.1     .05       0
Bank Sta=4993.2,5004.3
XS Rating Curve= 0 ,0
Exp/Cntr=0.3,0.1

Type RM Length L Ch R = 1 ,15424   ,240,240,240
BEGIN DESCRIPTION:
Mapping XS 97f829cd
END DESCRIPTION:
XS GIS Cut Line= 3
       2514077.3     13464432.59      2513181.44     13463807.58
      2512209.64     13463370.26
#Sta/Elev= 30
  3915.7   184.7  3966.9  184.68  4264.6  175.51    4411  171.44  4427.8  169.36
  4499.6  168.71  4784.2  157.17  4884.7  158.74  4920.4  156.52  4956.2  157.25
  4964.9  156.74  4979.3  152.81  5000.4  145.08  5000.9  144.58  5011.5  145.08
    5029  154.44    5059  158.69    5104  159.18  5173.4  156.59  5317.8  161.98
  5444.6  161.53  5490.8  163.33  5508.5  165.39    5514  164.06  5537.1   165.8
  5542.6  164.51  5565.7  164.27    5612  165.09    5924  174.61  6073.7  177.22
#Mann= 7 ,-1 , 0
  3915.7    .035       0  4264.6     .07       0  4427.8    .035       0
  4499.6     .12       0  5000.4     .05       0  5011.5     .12       0
  5444.6     .05       0
Bank Sta=5000.4,5011.5
XS Rating Curve= 0 ,0
Exp/Cntr=0.3,0.1
